HEC-RAS study South Fork.prj: South Fork Limited Detail Study

--- South Fork.g01 (geometry) --- (continued)

Type RM Length L Ch R = 1,81534,300,300,300
BEGIN DESCRIPTION:
South Fork 272.0
END DESCRIPTION:
XS GIS Cut Line= 4
      1429845.18       965294.77      1429362.52       965291.30
      1429232.29       965297.86      1429161.12       965286.09
#Sta/Elev= 30
  4472.5 1451.75  4508.7 1438.84  4522.4 1434.61  4539.1 1431.11  4572.8 1425.38
  4585.9 1422.42  4597.1 1422.73  4609.8 1425.26  4631.6 1425.71  4689.0 1424.45
  4780.5 1423.57  4807.1 1423.92  4833.7 1423.55  4842.0 1423.07  4896.9 1422.56
  4957.0 1422.93  4966.4 1422.95  4979.8 1422.11  4992.4 1421.84  4996.1 1421.00
  4997.6 1414.66  5002.4 1414.66  5003.9 1421.00  5032.0 1422.52  5044.9 1422.59
  5048.4 1422.25  5085.6 1424.74  5109.1 1432.65  5122.7 1443.04  5157.7 1446.21
#Mann=4,-1,0
  4472.5    0.08       0  4957.0    0.14       0  4996.1    0.05       0
  5003.9    0.14       0
#XS Ineff=2,0
    0.00 4900.00 1452.00               0
Permanent Ineff=
       F       F
Bank Sta=4996.1,5003.9
XS Rating Curve= 0
Exp/Cntr=0.3,0.1

Type RM Length L Ch R = 1,81234,240,240,240
BEGIN DESCRIPTION:
South Fork 271.0
END DESCRIPTION:
XS GIS Cut Line= 3
      1429893.81       965076.02      1429421.55       965069.08
      1429173.31       965077.75
#Sta/Elev= 30
  4455.7 1444.06  4468.6 1440.79  4478.1 1439.11  4489.8 1437.57  4544.7 1428.41
  4589.5 1421.84  4628.6 1416.97  4639.5 1416.42  4641.7 1415.83  4665.4 1417.89
  4721.6 1419.67  4757.9 1419.14  4798.4 1419.30  4814.3 1418.68  4841.7 1419.19
  4862.7 1418.74  4909.5 1419.27  4940.9 1418.39  4981.6 1418.35  4993.0 1413.03
  4995.7 1410.03  5004.3 1410.03  5007.0 1413.03  5010.6 1413.03  5017.6 1420.70
  5023.1 1423.54  5064.6 1428.30  5127.8 1434.51  5156.6 1439.43  5176.4 1443.44
#Mann=4,-1,0
  4455.7    0.08       0  4981.6    0.14       0  4993.0    0.05       0
  5007.0    0.14       0
#XS Ineff=2,0
    0.00 4750.00 1421.00               0
Permanent Ineff=
       F       F
Bank Sta=4993,5007
XS Rating Curve= 0
Exp/Cntr=0.3,0.1

Type RM Length L Ch R = 1,80994,249,249,249
BEGIN DESCRIPTION:
South Fork 270.0
END DESCRIPTION:
XS GIS Cut Line= 3
      1429923.29       964951.02      1429440.64       964860.74
      1429216.72       964813.87
#Sta/Elev= 30
  4513.9 1441.05  4528.1 1435.91  4547.3 1430.21  4572.8 1424.92  4594.7 1422.29
  4665.4 1416.16  4707.7 1415.24  4739.1 1413.90  4766.0 1415.45  4781.2 1415.68
  4869.8 1415.16  4903.5 1415.78  4926.5 1415.46  4959.8 1416.53  4965.2 1415.02
  4973.1 1412.66  4996.1 1411.11  4997.6 1408.11  5002.4 1408.11  5003.9 1411.11
  5004.9 1412.87  5013.0 1415.00  5048.8 1416.43  5068.7 1422.46  5114.3 1427.17
  5137.1 1430.85  5154.6 1431.11  5177.6 1435.01  5223.5 1439.11  5233.7 1440.50
#Mann=4,-1,0
  4513.9    0.08       0  4965.2    0.14       0  4996.1    0.05       0
  5003.9    0.14       0
#XS Ineff=2,0
    0.00 4900.00 1420.00               0
Permanent Ineff=
       F       F
Bank Sta=4996.1,5003.9
XS Rating Curve= 0
Exp/Cntr=0.3,0.1

Type RM Length L Ch R = 1,80745,228,228,228
BEGIN DESCRIPTION:
South Fork 269.0
END DESCRIPTION:
XS GIS Cut Line= 3
      1429926.75       964685.39      1429812.17       964678.45
      1429246.23       964661.09
#Sta/Elev= 30
  4532.0 1439.46  4572.7 1426.25  4591.9 1420.69  4607.0 1417.45  4661.0 1410.12
  4697.0 1410.38  4730.6 1412.26  4740.3 1410.75  4786.7 1411.65  4819.4 1410.43
  4945.4 1413.53  4959.9 1413.10  4972.7 1414.15  4974.9 1413.16  4993.0 1408.69
  4995.7 1404.80  5004.3 1404.80  5007.0 1407.80  5014.2 1409.55  5024.1 1409.76
  5049.2 1414.47  5061.6 1414.80  5075.5 1417.41  5083.4 1423.15  5089.8 1426.64
  5101.4 1431.62  5108.1 1430.94  5129.7 1432.51  5172.6 1436.26  5213.0 1440.83
#Mann=4,-1,0
  4532.0    0.08       0  4974.9    0.14       0  4993.0    0.05       0
  5007.0    0.14       0
#XS Ineff=2,0
    0.00 4897.00 1415.00               0
Permanent Ineff=
       F       F
Bank Sta=4993,5007
XS Rating Curve= 0
Exp/Cntr=0.5,0.3

Type RM Length L Ch R = 1,80517,32,32,32
BEGIN DESCRIPTION:
Private Bridge 2 US
END DESCRIPTION:
XS GIS Cut Line= 4
      1429842.22       964629.70      1429622.62       964609.20
      1429550.90       964426.23      1429413.26       964396.94
#Sta/Elev= 30
  4686.3 1414.83  4706.8 1412.38  4733.0 1410.53  4751.6 1407.97  4757.2 1407.83
  4762.3 1407.08  4782.0 1406.39  4787.0 1406.86  4806.1 1405.93  4812.9 1406.66
  4823.5 1408.71  4829.2 1409.16  4872.6 1409.03  4906.9 1409.91  4963.3 1410.03
  4971.5 1409.73  4991.6 1405.31  4994.0 1403.94  4995.0 1401.65  5005.0 1401.65
  5006.0 1403.94  5006.4 1408.24  5025.3 1410.07  5064.5 1410.27  5111.4 1412.02
  5134.1 1414.20  5151.0 1414.96  5178.8 1417.64  5234.1 1423.94  5244.1 1425.33
#Mann=4,-1,0
  4686.3    0.08       0  4994.0    0.05       0  5006.0    0.08       0
  5234.1    0.14       0
#XS Ineff=3,-1
 4691.20 4824.00 1412.02 4875.30 4990.00 1410.00 5010.00 5035.90 1410.00
Permanent Ineff=
       F       F       F
Bank Sta=4994,5006
XS Rating Curve= 0
Exp/Cntr=0.5,0.3

Type RM Length L Ch R =3,80503,,,
BEGIN DESCRIPTION:
Private Bridge 2 TOR
Structure ID: LDS_SF_B
Approximate Survey Structure
END DESCRIPTION:
Bridge Culvert--1,0,-1,-1,0
Deck Dist Width WeirC Skew NumUp NumDn MinLoCord MaxHiCord MaxSubmerge Is_Ogee
3,22,3,, 53, 53,,,0.95,0,1,1,,,
  4688.2  4710.4  4716.9  4728.8  4735.5  4748.7  4758.6  4758.7  4771.0  4784.6
  4796.9  4806.6  4810.9  4815.0  4822.3  4826.2  4829.4  4832.1  4837.5  4843.6
  4847.5  4855.4  4857.3  4869.0  4883.0  4923.3  4979.0  4979.0  5021.0  5021.0
  5061.7  5077.6  5093.0  5098.2  5108.7  5114.4  5120.1  5129.9  5137.4  5142.8
  5155.1  5159.7  5163.3  5165.1  5190.5  5202.4  5209.7  5222.0  5228.6  5238.7
  5251.5  5257.4  5277.7
 1414.17 1413.57 1412.66 1411.64 1411.22 1409.64 1408.22 1408.74 1406.75 1405.86
 1403.97 1404.70 1405.29 1405.15 1405.24 1405.71 1404.91 1405.40 1407.23 1405.71
 1405.52 1406.56 1406.57 1407.53 1408.56 1410.00 1410.00 1410.00 1410.00 1410.00
 1410.00 1410.53 1410.33 1410.66 1410.82 1411.03 1411.58 1411.94 1412.58 1413.19
 1413.90 1414.01 1414.43 1414.75 1416.64 1417.79 1418.67 1419.50 1420.22 1421.66
 1423.31 1424.55 1427.27
 1381.65 1381.65 1381.65 1381.65 1381.65 1381.65 1381.65 1381.65 1381.65 1381.65
 1381.65 1381.65 1381.65 1381.65 1381.65 1381.65 1381.65 1381.65 1381.65 1381.65
 1381.65 1381.65 1381.65 1381.65 1381.65 1381.65 1381.65 1408.50 1408.50 1381.65
 1381.65 1381.65 1381.65 1381.65 1381.65 1381.65 1381.65 1381.65 1381.65 1381.65
 1381.65 1381.65 1381.65 1381.65 1381.65 1381.65 1381.65 1381.65 1381.65 1381.65
 1381.65 1381.65 1381.65
  4688.2  4710.4  4716.9  4728.8  4735.5  4748.7  4758.6  4758.7  4771.0  4784.6
  4796.9  4806.6  4810.9  4815.0  4822.3  4826.2  4829.4  4832.1  4837.5  4843.6
  4847.5  4855.4  4857.3  4869.0  4883.0  4923.3  4979.0  4979.0  5021.0  5021.0
  5061.7  5077.6  5093.0  5098.2  5108.7  5114.4  5120.1  5129.9  5137.4  5142.8
  5155.1  5159.7  5163.3  5165.1  5190.5  5202.4  5209.7  5222.0  5228.6  5238.7
  5251.5  5257.4  5277.7
 1414.17 1413.57 1412.66 1411.64 1411.22 1409.64 1408.22 1408.74 1406.75 1405.86
 1403.97 1404.70 1405.29 1405.15 1405.24 1405.71 1404.91 1405.40 1407.23 1405.71
 1405.52 1406.56 1406.57 1407.53 1408.56 1410.00 1410.00 1410.00 1410.00 1410.00
 1410.00 1410.53 1410.33 1410.66 1410.82 1411.03 1411.58 1411.94 1412.58 1413.19
 1413.90 1414.01 1414.43 1414.75 1416.64 1417.79 1418.67 1419.50 1420.22 1421.66
 1423.31 1424.55 1427.27
 1381.65 1381.65 1381.65 1381.65 1381.65 1381.65 1381.65 1381.65 1381.65 1381.65
 1381.65 1381.65 1381.65 1381.65 1381.65 1381.65 1381.65 1381.65 1381.65 1381.65
 1381.65 1381.65 1381.65 1381.65 1381.65 1381.65 1381.65 1408.50 1408.50 1381.65
 1381.65 1381.65 1381.65 1381.65 1381.65 1381.65 1381.65 1381.65 1381.65 1381.65
 1381.65 1381.65 1381.65 1381.65 1381.65 1381.65 1381.65 1381.65 1381.65 1381.65
 1381.65 1381.65 1381.65
BR Coef=1,1,0,1.25,0,,,0.8,0,2,0,
WSPro=,,,, 1 ,,,, 0 ,,,, 0 ,,,,-1 ,-1 ,-1 , 0 , 0 , 0 , 0 , 0
BC Design=,,0,,0,,,,,,

Type RM Length L Ch R = 1,80485,291,291,291
BEGIN DESCRIPTION:
Private Bridge 2 DS
END DESCRIPTION:
XS GIS Cut Line= 4
      1429845.14       964594.56      1429640.19       964579.92
      1429587.49       964404.27      1429420.62       964367.68
#Sta/Elev= 30
  4722.6 1414.40  4728.1 1413.06  4739.0 1411.59  4771.6 1408.22  4782.4 1406.62
  4785.0 1405.53  4822.0 1406.01  4838.1 1407.32  4847.6 1406.17  4856.0 1407.54
  4862.7 1406.92  4892.6 1407.25  4906.0 1408.94  4951.9 1408.88  4973.6 1409.48
  4983.6 1408.19  4994.0 1402.56  4995.0 1401.40  5005.0 1401.40  5006.0 1402.56
  5022.7 1409.61  5083.1 1409.39  5125.4 1410.58  5170.4 1413.31  5215.8 1416.89
  5222.3 1417.84  5239.0 1418.72  5261.8 1421.53  5270.7 1423.52  5282.3 1426.09
#Mann=4,-1,0
  4722.6    0.08       0  4994.0    0.05       0  5006.0    0.08       0
  5270.7    0.14       0
#XS Ineff=3,-1
 4739.50 4824.00 1410.78 4902.30 4989.60 1408.00 5010.00 5062.00 1408.00
Permanent Ineff=
       F       F       F
Bank Sta=4994,5006
XS Rating Curve= 0
Exp/Cntr=0.5,0.3

Type RM Length L Ch R = 1,80194,292,292,292
BEGIN DESCRIPTION:
South Fork 268.0
END DESCRIPTION:
XS GIS Cut Line= 5
      1429938.98       964516.31      1429888.62       964495.47
      1429770.57       964301.02      1429629.94       964276.72
      1429511.89       964259.36
#Sta/Elev= 30
  4839.7 1433.80  4849.6 1431.10  4893.3 1420.02  4902.9 1417.83  4921.5 1414.13
  4939.5 1408.73  4958.8 1406.60  4967.9 1409.03  4978.4 1409.37  4988.6 1400.36
  4992.2 1400.28  4995.2 1398.28  5004.8 1398.28  5007.8 1400.28  5016.3 1404.04
  5035.6 1405.28  5131.3 1404.72  5144.2 1405.05  5170.4 1406.38  5183.9 1406.20
  5207.4 1406.69  5223.3 1406.71  5253.6 1407.27  5265.5 1407.71  5277.6 1408.29
  5302.3 1410.13  5321.3 1411.82  5350.0 1414.87  5367.0 1416.41  5383.7 1417.54
#Mann=3,-1,0
  4839.7    0.08       0  4992.2    0.05       0  5007.8    0.08       0
#XS Ineff=2,0
       0                 5035.60    0.00 1410.00
Permanent Ineff=
       F       F
Bank Sta=4992.2,5007.8
XS Rating Curve= 0
Exp/Cntr=0.5,0.3

Type RM Length L Ch R = 1,79902,41,41,41
BEGIN DESCRIPTION:
Private Culvert 3
END DESCRIPTION:
XS GIS Cut Line= 4
      1430127.29       964137.93      1430063.55       964114.45
      1429782.72       964266.30      1429522.29       964222.90
#Sta/Elev= 30
  4815.6 1426.81  4830.2 1424.70  4883.5 1411.11  4896.0 1411.18  4909.7 1412.66
  4916.8 1412.64  4923.7 1412.00  4939.0 1409.77  4948.8 1407.98  4963.6 1404.34
  4977.2 1401.79  4993.7 1399.18  4995.5 1394.00  5004.5 1394.00  5006.3 1399.18
  5014.3 1400.48  5035.1 1400.51  5081.4 1402.28  5132.9 1401.79  5158.0 1403.06
  5235.8 1404.65  5248.6 1405.30  5268.3 1405.41  5289.4 1406.10  5303.1 1405.89
  5338.5 1406.43  5390.3 1409.52  5414.7 1411.64  5433.8 1413.91  5466.8 1416.57
#Mann=3,-1,0
  4815.6    0.08       0  4993.7    0.05       0  5006.3    0.08       0
#XS Ineff=3,-1
 4943.00 4993.00 1400.00 5007.00 5057.00 1400.00 5106.20 5383.20 1407.87
Permanent Ineff=
       F       F       F
Bank Sta=4993.7,5006.3
XS Rating Curve= 0
Exp/Cntr=0.5,0.3

Type RM Length L Ch R =2,79882,,,
BEGIN DESCRIPTION:
Private Culvert 3 TOR
Structure ID: LDS_SF_C
Approximate Survey Structure
END DESCRIPTION:
Bridge Culvert--1,0,-1,-1,0
Deck Dist Width WeirC Skew NumUp NumDn MinLoCord MaxHiCord MaxSubmerge Is_Ogee
2.5,35,3,, 56, 56,,,0.95,0,1,1,,,
  4768.5  4790.4  4806.8  4828.4  4832.8  4851.0  4859.6  4871.1  4876.7  4887.6
  4891.5  4905.4  4908.9  4939.7  4945.4  4955.8  4958.8  4965.9  4970.8  5007.0
  5008.2  5019.9  5026.3  5040.9  5043.7  5065.0  5076.7  5084.5  5099.7  5110.9
  5143.4  5146.7  5167.5  5182.3  5193.8  5205.7  5219.5  5242.7  5259.3  5265.9
  5273.3  5312.0  5314.8  5329.6  5336.1  5345.4  5359.0  5372.9  5385.1  5399.6
  5406.0  5412.5  5418.9  5429.5  5450.7  5452.5
 1426.97 1426.60 1424.38 1418.90 1417.33 1412.07 1410.88 1407.42 1406.35 1405.99
 1405.78 1405.50 1405.85 1404.67 1403.94 1402.30 1401.92 1400.28 1400.00 1400.00
 1400.12 1400.23 1400.41 1401.00 1401.05 1400.72 1401.40 1401.66 1401.52 1401.64
 1402.68 1402.92 1403.79 1404.12 1404.23 1404.04 1404.40 1405.14 1405.18 1405.43
 1405.58 1405.54 1405.68 1406.93 1407.34 1407.60 1408.20 1408.99 1409.90 1411.14
 1411.82 1412.68 1413.41 1414.49 1415.65 1415.91
 1374.00 1374.00 1374.00 1374.00 1374.00 1374.00 1374.00 1374.00 1374.00 1374.00
 1374.00 1374.00 1374.00 1374.00 1374.00 1374.00 1374.00 1374.00 1374.00 1374.00
 1374.00 1374.00 1374.00 1374.00 1374.00 1374.00 1374.00 1374.00 1374.00 1374.00
 1374.00 1374.00 1374.00 1374.00 1374.00 1374.00 1374.00 1374.00 1374.00 1374.00
 1374.00 1374.00 1374.00 1374.00 1374.00 1374.00 1374.00 1374.00 1374.00 1374.00
 1374.00 1374.00 1374.00 1374.00 1374.00 1374.00
  4768.5  4790.4  4806.8  4828.4  4832.8  4851.0  4859.6  4871.1  4876.7  4887.6
  4891.5  4905.4  4908.9  4939.7  4945.4  4955.8  4958.8  4965.9  4970.8  5007.0
  5008.2  5019.9  5026.3  5040.9  5043.7  5065.0  5076.7  5084.5  5099.7  5110.9
  5143.4  5146.7  5167.5  5182.3  5193.8  5205.7  5219.5  5242.7  5259.3  5265.9
  5273.3  5312.0  5314.8  5329.6  5336.1  5345.4  5359.0  5372.9  5385.1  5399.6
  5406.0  5412.5  5418.9  5429.5  5450.7  5452.5
 1426.97 1426.60 1424.38 1418.90 1417.33 1412.07 1410.88 1407.42 1406.35 1405.99
 1405.78 1405.50 1405.85 1404.67 1403.94 1402.30 1401.92 1400.28 1400.00 1400.00
 1400.12 1400.23 1400.41 1401.00 1401.05 1400.72 1401.40 1401.66 1401.52 1401.64
 1402.68 1402.92 1403.79 1404.12 1404.23 1404.04 1404.40 1405.14 1405.18 1405.43
 1405.58 1405.54 1405.68 1406.93 1407.34 1407.60 1408.20 1408.99 1409.90 1411.14
 1411.82 1412.68 1413.41 1414.49 1415.65 1415.91
 1373.83 1373.83 1373.83 1373.83 1373.83 1373.83 1373.83 1373.83 1373.83 1373.83
 1373.83 1373.83 1373.83 1373.83 1373.83 1373.83 1373.83 1373.83 1373.83 1373.83
 1373.83 1373.83 1373.83 1373.83 1373.83 1373.83 1373.83 1373.83 1373.83 1373.83
 1373.83 1373.83 1373.83 1373.83 1373.83 1373.83 1373.83 1373.83 1373.83 1373.83
 1373.83 1373.83 1373.83 1373.83 1373.83 1373.83 1373.83 1373.83 1373.83 1373.83
 1373.83 1373.83 1373.83 1373.83 1373.83 1373.83
Culvert=1,4,,35,0.024,0.9,1,2,3,1394,5000,1393.83,5000,Culvert #1,0,2.5
Culvert Bottom n=0.024
Culvert Bottom Depth=0
Culvert Depth Blocked=0
BC Design=,,0,,0,,,,,,

Type RM Length L Ch R = 1,79861,313,313,313
BEGIN DESCRIPTION:
Private Culvert 3 DS
END DESCRIPTION:
XS GIS Cut Line= 4
      1430146.32       964112.20      1430061.16       964081.16
      1429753.20       964221.16      1429527.49       964186.44
#Sta/Elev= 30
  4773.5 1425.97  4791.0 1423.15  4812.1 1418.79  4835.6 1410.43  4857.8 1407.41
  4872.2 1404.67  4882.8 1404.73  4907.9 1402.78  4931.5 1401.71  4960.4 1399.10
  4980.6 1399.17  4984.7 1398.24  4993.0 1395.18  4995.0 1393.83  5005.0 1393.83
  5007.0 1395.18  5009.7 1397.92  5021.5 1400.11  5055.6 1400.29  5089.7 1401.19
  5118.5 1402.92  5145.0 1403.69  5193.8 1403.97  5219.7 1404.88  5288.4 1405.70
  5321.0 1407.14  5369.0 1410.33  5393.1 1413.22  5417.2 1414.93  5430.8 1416.59
#Mann=3,-1,0
  4773.5    0.08       0  4993.0    0.05       0  5007.0    0.08       0
#XS Ineff=2,0
    0.00 4993.00 1400.00 5007.00    0.00 1400.00
Permanent Ineff=
       F       F
Bank Sta=4993,5007
XS Rating Curve= 0
Exp/Cntr=0.5,0.3

Type RM Length L Ch R = 1,79548,308,308,308
BEGIN DESCRIPTION:
South Fork 265.0
END DESCRIPTION:
XS GIS Cut Line= 3
      1430251.38       963895.46      1429863.39       963873.63
      1429589.94       963852.06
#Sta/Elev= 30
  4611.4 1421.95  4627.8 1419.99  4644.2 1415.89  4653.0 1413.57  4677.7 1403.68
  4703.3 1398.09  4738.6 1396.95  4776.3 1396.84  4801.0 1396.32  4846.7 1396.98
  4860.9 1396.21  4893.4 1396.22  4917.0 1396.67  4933.9 1395.66  4940.4 1393.59
  4965.1 1390.44  4990.0 1392.43  4994.5 1389.32  4996.6 1386.32  5003.4 1386.32
  5005.5 1389.32  5006.4 1391.75  5022.6 1395.90  5038.9 1398.49  5063.6 1398.32
  5174.8 1401.25  5216.8 1403.67  5250.2 1406.73  5263.3 1408.62  5274.3 1411.63
#Mann=4,-1,0
  4611.4    0.08       0  4994.5    0.05       0  5005.5    0.08       0
  5250.2    0.14       0
Bank Sta=4994.5,5005.5
XS Rating Curve= 0
Exp/Cntr=0.3,0.1

Type RM Length L Ch R = 1,79240,278,278,278
BEGIN DESCRIPTION:
South Fork 264.0
END DESCRIPTION:
XS GIS Cut Line= 3
      1430237.53       963680.19      1430030.92       963607.27
      1429642.04       963560.40
#Sta/Elev= 30
  4684.2 1408.60  4746.8 1406.47  4762.5 1406.30  4767.9 1405.62  4775.5 1405.73
  4798.3 1404.88  4809.9 1403.89  4815.4 1402.60  4831.9 1400.55  4854.0 1394.54
  4874.6 1386.62  4883.7 1387.20  4901.7 1386.34  4921.5 1387.77  4944.5 1387.41
  4969.2 1387.88  4974.2 1387.73  4989.9 1385.33  4996.1 1384.93  4997.6 1381.93
  5002.4 1381.93  5003.9 1384.93  5035.3 1390.26  5056.4 1390.65  5077.6 1390.33
  5141.7 1392.32  5187.5 1394.82  5227.3 1397.64  5267.7 1402.19  5295.0 1405.72
#Mann=4,-1,0
  4684.2    0.08       0  4996.1    0.05       0  5003.9    0.08       0
  5267.7    0.14       0
Bank Sta=4996.1,5003.9
XS Rating Curve= 0
Exp/Cntr=0.3,0.1

Type RM Length L Ch R = 1,78962,311,311,311
BEGIN DESCRIPTION:
South Fork 263.0
END DESCRIPTION:
XS GIS Cut Line= 4
      1430331.24       963501.35      1430185.43       963376.37
      1429834.94       963350.99      1429680.26       963355.53
#Sta/Elev= 30
  4506.1 1411.72  4533.8 1408.81  4595.8 1403.21  4621.5 1399.62  4637.3 1396.52
  4657.9 1393.31  4698.1 1389.09  4726.3 1386.80  4751.7 1386.05  4797.2 1385.98
  4827.7 1386.27  4844.7 1385.96  4872.4 1386.66  4914.9 1386.72  4966.1 1384.36
  4977.0 1381.94  4983.6 1381.68  4994.2 1380.06  4996.4 1377.06  5003.6 1377.06
  5005.9 1379.00  5010.9 1380.03  5021.7 1385.04  5048.0 1387.64  5079.5 1391.55
  5144.0 1401.35  5154.7 1402.85  5176.9 1405.06  5198.7 1411.75  5204.3 1414.49
#Mann=4,-1,0
  4506.1    0.08       0  4994.2    0.05       0  5005.9    0.08       0
  5144.0    0.14       0
Bank Sta=4994.2,5005.9
XS Rating Curve= 0
Exp/Cntr=0.3,0.1

Type RM Length L Ch R = 1,78651,300,300,300
BEGIN DESCRIPTION:
South Fork 262.0
END DESCRIPTION:
XS GIS Cut Line= 3
      1430319.08       963388.49      1430220.16       963296.51
      1429831.23       962964.88
#Sta/Elev= 30
  4512.3 1402.05  4556.4 1395.84  4578.9 1392.18  4620.5 1387.54  4660.1 1384.75
  4710.7 1383.28  4746.5 1382.89  4785.7 1382.52  4821.2 1383.05  4829.6 1382.72
  4837.2 1381.78  4853.9 1381.97  4869.2 1380.60  4975.9 1380.40  4992.1 1378.25
  4996.1 1376.29  4997.6 1373.29  5002.4 1373.29  5003.9 1376.29  5018.6 1379.86
  5062.2 1381.44  5077.0 1381.08  5095.2 1384.55  5099.3 1385.55  5105.1 1387.77
  5118.9 1394.48  5134.8 1419.22  5142.8 1431.11  5154.0 1439.78  5158.5 1442.78
#Mann=4,-1,0
  4512.3    0.08       0  4996.1    0.05       0  5003.9    0.08       0
  5062.2    0.14       0
#XS Ineff=2,0
    0.00 4901.40 1390.18 5056.60    0.00 1389.90
Permanent Ineff=
       F       F
Bank Sta=4996.1,5003.9
XS Rating Curve= 0
Exp/Cntr=0.3,0.1

Type RM Length L Ch R = 1,78351,280,280,280
BEGIN DESCRIPTION:
South Fork 261.0
END DESCRIPTION:
XS GIS Cut Line= 5
      1430334.74       963374.64      1430294.48       963094.66
      1430235.78       962999.63      1430150.85       962909.12
      1430011.79       962822.52
#Sta/Elev= 30
  4586.8 1400.59  4615.9 1395.38  4657.9 1392.48  4666.7 1390.93  4698.6 1387.99
  4765.1 1382.96  4810.7 1381.26  4852.7 1380.24  4882.5 1380.03  4892.2 1379.28
  4907.8 1378.97  4932.6 1377.52  4980.2 1375.62  4988.6 1375.81  4996.1 1372.53
  4997.6 1369.53  5002.4 1369.53  5003.9 1372.53  5009.3 1375.13  5014.5 1376.88
  5020.5 1377.34  5061.0 1376.76  5105.0 1378.12  5125.2 1380.63  5140.4 1380.80
  5167.8 1382.71  5220.5 1388.00  5250.6 1392.00  5264.1 1394.98  5269.3 1397.08
#Mann=4,-1,0
  4586.8    0.08       0  4996.1    0.05       0  5003.9    0.08       0
  5220.5    0.14       0
Bank Sta=4996.1,5003.9
XS Rating Curve= 0
Exp/Cntr=0.3,0.1

Type RM Length L Ch R = 1,78071,332,332,332
BEGIN DESCRIPTION:
South Fork 260.0
END DESCRIPTION:
XS GIS Cut Line= 4
      1430610.68       963103.43      1430590.70       963005.35
      1430246.20       962801.71      1430048.30       962680.20
#Sta/Elev= 30
  4484.5 1393.76  4504.9 1394.24  4543.4 1386.79  4571.1 1383.80  4654.7 1378.63
  4716.9 1377.21  4782.1 1374.07  4803.8 1374.14  4823.9 1375.04  4824.0 1374.51
  4856.8 1372.01  4864.5 1374.52  4889.8 1374.64  4907.3 1369.68  4921.7 1370.85
  4940.6 1370.38  4947.3 1371.76  4975.5 1373.39  4982.5 1373.02  4994.2 1369.55
  4996.4 1366.55  5003.6 1366.55  5005.9 1368.40  5011.3 1369.20  5028.3 1378.30
  5044.3 1379.53  5092.8 1387.84  5155.4 1395.34  5213.0 1403.13  5217.0 1404.13
#Mann=4,-1,0
  4484.5    0.08       0  4994.2    0.05       0  5005.9    0.08       0
  5155.4    0.14       0
#XS Ineff=2,0
    0.00 4889.10 1380.81               0
Permanent Ineff=
       F       F
Bank Sta=4994.2,5005.9
XS Rating Curve= 0
Exp/Cntr=0.3,0.1

Type RM Length L Ch R = 1,77739,323,323,323
BEGIN DESCRIPTION:
South Fork 259.0
END DESCRIPTION:
XS GIS Cut Line= 4
      1430721.90       962947.55      1430570.44       962851.47
      1430518.77       962584.70      1430306.95       962442.33
#Sta/Elev= 30
  4695.8 1393.07  4708.5 1388.50  4730.1 1387.73  4744.5 1383.57  4772.6 1380.38
  4785.8 1379.68  4826.3 1378.74  4867.7 1376.42  4908.3 1374.72  4977.7 1370.67
  4990.4 1368.98  4995.4 1367.20  4996.9 1364.20  5003.1 1364.20  5004.6 1367.20
  5005.8 1369.66  5019.6 1373.60  5021.8 1373.41  5029.3 1370.67  5032.6 1370.78
  5053.9 1369.43  5114.5 1368.82  5208.0 1371.62  5254.4 1371.99  5282.6 1373.10
  5309.8 1374.76  5345.6 1377.99  5371.1 1381.77  5383.3 1383.58  5402.1 1388.18
#Mann=4,-1,0
  4695.8    0.08       0  4995.4    0.05       0  5004.6    0.08       0
  5371.1    0.14       0
#XS Ineff=2,0
       0                 5021.30    0.00 1374.68
Permanent Ineff=
       F       F
Bank Sta=4995.4,5004.6
XS Rating Curve= 0
Exp/Cntr=0.3,0.1

Type RM Length L Ch R = 1,77416,281,281,281
BEGIN DESCRIPTION:
South Fork 258.0
END DESCRIPTION:
XS GIS Cut Line= 3
      1430970.15       962645.46      1430708.00       962537.83
      1430352.10       962395.46
#Sta/Elev= 30
  4694.9 1385.00  4721.7 1378.42  4733.8 1376.27  4741.2 1373.98  4776.7 1371.64
  4805.5 1370.61  4819.9 1369.64  4909.1 1369.78  4922.6 1369.43  4965.4 1366.85
  4972.2 1367.20  4978.3 1363.56  4995.4 1359.74  4996.9 1356.74  5003.1 1356.74
  5004.6 1359.74  5009.9 1362.67  5015.7 1366.57  5030.8 1366.64  5038.5 1367.68
  5059.8 1368.72  5080.3 1368.98  5139.4 1368.11  5191.5 1368.89  5212.0 1369.59
  5275.6 1373.62  5296.5 1375.80  5322.7 1379.03  5339.8 1381.53  5361.6 1387.01
#Mann=4,-1,0
  4694.9    0.08       0  4995.4    0.05       0  5004.6    0.08       0
  5322.7    0.14       0
Bank Sta=4995.4,5004.6
XS Rating Curve= 0
Exp/Cntr=0.3,0.1

Type RM Length L Ch R = 1,77135,300,300,300
BEGIN DESCRIPTION:
South Fork 257.0
END DESCRIPTION:
XS GIS Cut Line= 3
      1431076.03       962482.25      1430802.09       962283.58
      1430581.24       962129.82
#Sta/Elev= 30
  4661.6 1375.52  4668.9 1376.03  4683.1 1375.59  4691.1 1373.63  4726.1 1371.37
  4755.1 1370.08  4768.5 1368.95  4857.6 1366.55  4878.5 1365.18  4933.1 1363.25
  4940.8 1362.59  4955.9 1360.16  4980.7 1358.39  4995.4 1356.37  4996.9 1353.37
  5003.1 1353.37  5004.6 1356.37  5006.8 1357.15  5011.4 1359.74  5019.8 1363.70
  5039.9 1363.01  5061.0 1363.30  5080.5 1363.03  5087.4 1363.45  5100.0 1363.21
  5137.6 1364.40  5218.6 1368.53  5246.4 1370.79  5260.1 1372.61  5269.1 1374.21
#Mann=3,-1,0
  4661.6    0.08       0  4995.4    0.05       0  5004.6    0.08       0
Bank Sta=4995.4,5004.6
XS Rating Curve= 0
Exp/Cntr=0.3,0.1

Type RM Length L Ch R = 1,76835,317,317,317
BEGIN DESCRIPTION:
South Fork 256.0
END DESCRIPTION:
XS GIS Cut Line= 3
      1431289.62       962247.90      1430991.12       962064.58
      1430794.85       961937.16
#Sta/Elev= 30
  4649.7 1375.60  4652.8 1374.97  4662.5 1374.18  4678.1 1371.74  4710.6 1367.93
  4732.4 1367.29  4761.8 1364.68  4836.6 1360.62  4864.4 1360.41  4917.6 1357.75
  4925.3 1357.86  4957.7 1356.50  4979.3 1356.11  4987.4 1355.19  4995.4 1352.17
  4996.9 1349.17  5003.1 1349.17  5004.6 1352.17  5013.9 1355.50  5021.8 1357.36
  5030.7 1358.48  5052.5 1359.24  5126.1 1358.99  5145.7 1359.36  5160.5 1360.57
  5168.6 1361.12  5175.8 1362.10  5188.5 1366.17  5223.8 1386.99  5234.0 1392.31
#Mann=4,-1,0
  4649.7    0.08       0  4995.4    0.05       0  5004.6    0.08       0
  5160.5    0.14       0
Bank Sta=4995.4,5004.6
XS Rating Curve= 0
Exp/Cntr=0.3,0.1

Type RM Length L Ch R = 1,76518,83,83,83
BEGIN DESCRIPTION:
South Fork 255.0
END DESCRIPTION:
XS GIS Cut Line= 3
      1431492.77       961978.82      1431187.17       961817.34
      1430923.26       961674.97
#Sta/Elev= 30
  4640.1 1379.06  4647.1 1376.89  4655.8 1377.33  4668.0 1376.14  4675.9 1371.94
  4688.5 1367.87  4709.8 1364.65  4718.8 1362.72  4753.4 1360.31  4783.7 1358.59
  4867.9 1356.05  4919.4 1354.17  4948.6 1353.71  4960.8 1353.93  4980.6 1350.80
  4995.4 1346.92  4996.9 1343.92  5003.1 1343.92  5004.6 1346.92  5023.6 1352.97
  5068.0 1353.38  5096.6 1354.25  5108.6 1354.01  5187.4 1354.55  5206.1 1355.43
  5213.9 1356.05  5228.1 1357.76  5240.8 1359.46  5247.3 1360.88  5285.6 1377.49
#Mann=4,-1,0
  4640.1    0.08       0  4995.4    0.05       0  5004.6    0.08       0
  5228.1    0.14       0
Bank Sta=4995.4,5004.6
XS Rating Curve= 0
Exp/Cntr=0.5,0.3

Type RM Length L Ch R = 1,76435,27,27,27
BEGIN DESCRIPTION:
LDS_SFMR_08 US
END DESCRIPTION:
XS GIS Cut Line= 2
      1431531.26       961851.16      1430943.78       961642.89
#Sta/Elev= 30
  4662.6 1374.75  4677.0 1371.57  4686.2 1369.92  4698.8 1366.94  4721.1 1362.72
  4729.9 1362.16  4741.5 1360.49  4759.4 1358.86  4787.4 1357.20  4829.9 1355.47
  4851.3 1355.00  4888.9 1354.65  4912.6 1353.70  4939.9 1353.20  4957.7 1352.49
  4979.2 1350.61  4982.0 1347.99  4991.0 1343.10  5009.0 1343.10  5018.0 1347.99
  5040.5 1351.47  5063.1 1352.27  5085.1 1352.68  5093.6 1353.19  5167.1 1353.61
  5205.4 1354.92  5225.0 1356.43  5244.8 1359.18  5256.0 1361.48  5285.9 1372.51
#Mann=4,-1,0
  4662.6    0.08       0  4982.0    0.05       0  5018.0    0.08       0
  5244.8    0.14       0
#XS Ineff=2,0
    0.00 4976.80 1351.03 5023.10    0.00 1351.31
Permanent Ineff=
       F       F
Bank Sta=4982,5018
XS Rating Curve= 0
Exp/Cntr=0.5,0.3

Type RM Length L Ch R =3,76420,,,
BEGIN DESCRIPTION:
LDS_SFMR_08 TOR
Structure ID: LDS_SFMR_08
Approximate Survey Structure
END DESCRIPTION:
Bridge Culvert--1,0,-1,-1,0
Deck Dist Width WeirC Skew NumUp NumDn MinLoCord MaxHiCord MaxSubmerge Is_Ogee
6.5,17,3,,52,52,,,0.95,0,1,1,,,
  4661.2  4680.7  4684.2  4696.8  4706.2  4712.2  4728.1  4741.5  4750.7  4759.9
  4763.6  4785.2  4793.8  4806.8  4815.8  4828.4  4837.4  4841.0  4849.9  4858.8
  4870.5  4879.1  4889.1  4899.0  4906.8  4911.4  4917.0  4920.2  4933.0  4953.8
  4956.4  4961.9  4980.5  4983.3  4983.3  5016.8  5016.8  5175.2  5186.1  5193.7
  5196.3  5205.3  5217.1  5225.0  5233.5  5243.6  5245.5  5253.5  5260.8  5277.1
  5285.3  5297.6
 1374.91 1370.71 1370.03 1367.15 1365.65 1364.21 1361.54 1360.19 1359.04 1358.34
 1358.00 1356.62 1356.33 1355.64 1355.39 1354.86 1354.73 1354.62 1354.25 1354.40
 1353.98 1353.95 1353.74 1353.68 1353.55 1353.40 1353.30 1353.28 1352.90 1352.55
 1352.84 1352.75 1351.31 1351.31 1351.31 1351.31 1351.31 1351.30 1354.14 1354.45
 1354.53 1354.90 1355.54 1356.23 1357.15 1358.47 1358.77 1360.49 1362.34 1368.36
 1371.13 1374.94
 1323.10 1323.10 1323.10 1323.10 1323.10 1323.10 1323.10 1323.10 1323.10 1323.10
 1323.10 1323.10 1323.10 1323.10 1323.10 1323.10 1323.10 1323.10 1323.10 1323.10
 1323.10 1323.10 1323.10 1323.10 1323.10 1323.10 1323.10 1323.10 1323.10 1323.10
 1323.10 1323.10 1323.10 1323.10 1349.30 1349.30 1323.10 1323.10 1323.10 1323.10
 1323.10 1323.10 1323.10 1323.10 1323.10 1323.10 1323.10 1323.10 1323.10 1323.10
 1323.10 1323.10
  4661.2  4680.7  4684.2  4696.8  4706.2  4712.2  4728.1  4741.5  4750.7  4759.9
  4763.6  4785.2  4793.8  4806.8  4815.8  4828.4  4837.4  4841.0  4849.9  4858.8
  4870.5  4879.1  4889.1  4899.0  4906.8  4911.4  4917.0  4920.2  4933.0  4953.8
  4956.4  4961.9  4980.5  4983.3  4983.3  5016.8  5016.8  5175.2  5186.1  5193.7
  5196.3  5205.3  5217.1  5225.0  5233.5  5243.6  5245.5  5253.5  5260.8  5277.1
  5285.3  5297.6
 1374.91 1370.71 1370.03 1367.15 1365.65 1364.21 1361.54 1360.19 1359.04 1358.34
 1358.00 1356.62 1356.33 1355.64 1355.39 1354.86 1354.73 1354.62 1354.25 1354.40
 1353.98 1353.95 1353.74 1353.68 1353.55 1353.40 1353.30 1353.28 1352.90 1352.55
 1352.84 1352.75 1351.31 1351.31 1351.31 1351.31 1351.31 1351.30 1354.14 1354.45
 1354.53 1354.90 1355.54 1356.23 1357.15 1358.47 1358.77 1360.49 1362.34 1368.36
 1371.13 1374.94
 1323.10 1323.10 1323.10 1323.10 1323.10 1323.10 1323.10 1323.10 1323.10 1323.10
 1323.10 1323.10 1323.10 1323.10 1323.10 1323.10 1323.10 1323.10 1323.10 1323.10
 1323.10 1323.10 1323.10 1323.10 1323.10 1323.10 1323.10 1323.10 1323.10 1323.10
 1323.10 1323.10 1323.10 1323.10 1349.30 1349.30 1323.10 1323.10 1323.10 1323.10
 1323.10 1323.10 1323.10 1323.10 1323.10 1323.10 1323.10 1323.10 1323.10 1323.10
 1323.10 1323.10
Abutment Skew #Up #Dn=,2,2
  4983.3  4984.3
 1349.30 1347.53
  4983.3  4984.3
 1349.30 1347.08
Abutment Skew #Up #Dn=,2,2
  5015.8  5016.8
 1347.42 1349.30
  5015.8  5016.8
 1347.17 1349.30
BR Coef=1,1,0,1.25,0,,,0.8,0,2,0,
WSPro=,,,, 1 ,,,, 0 ,,,, 0 ,,,,-1 ,-1 ,-1 , 0 , 0 , 0 , 0 , 0
BC Design=,,0,,0,,,,,,

Type RM Length L Ch R = 1,76408,295,295,295
BEGIN DESCRIPTION:
LDS_SFMR_08 DS
END DESCRIPTION:
XS GIS Cut Line= 2
      1431544.26       961819.92      1430946.44       961622.09
#Sta/Elev= 30
  4665.6 1373.89  4674.7 1372.14  4684.0 1369.65  4706.0 1365.60  4719.0 1362.76
  4727.9 1361.33  4750.5 1358.95  4785.0 1356.46  4849.8 1353.87  4920.1 1352.91
  4953.8 1352.00  4961.9 1352.87  4988.1 1349.67  4990.0 1349.00  4995.0 1342.85
  5007.2 1342.85  5014.4 1349.00  5016.2 1349.13  5018.2 1350.19  5026.7 1351.04
  5039.8 1351.08  5093.2 1352.84  5167.0 1353.49  5205.5 1354.79  5225.0 1355.90
  5233.7 1356.77  5245.7 1358.23  5253.8 1360.24  5266.1 1363.26  5295.3 1372.30
#Mann=4,-1,0
  4665.6    0.08       0  4990.0    0.05       0  5014.4    0.08       0
  5253.8    0.14       0
#XS Ineff=2,0
    0.00 4976.80 1351.00 5023.10    0.00 1351.00
Permanent Ineff=
       F       F
Bank Sta=4990,5014.4
XS Rating Curve= 0
Exp/Cntr=0.5,0.3

Type RM Length L Ch R = 1,76113,217,217,217
BEGIN DESCRIPTION:
South Fork 254.0
END DESCRIPTION:
XS GIS Cut Line= 4
      1431635.12       961652.42      1431501.28       961587.75
      1431357.31       961480.53      1431199.36       961364.24
#Sta/Elev= 30
  4587.3 1373.63  4595.0 1373.43  4616.6 1368.76  4638.0 1365.14  4660.2 1360.65
  4673.3 1357.26  4681.9 1355.93  4723.9 1351.90  4745.1 1350.78  4785.8 1349.73
  4866.6 1349.39  4918.0 1347.66  4944.9 1347.19  4974.1 1347.73  4995.4 1341.80
  4996.9 1338.80  5003.1 1338.80  5004.6 1341.80  5009.7 1343.44  5015.1 1344.58
  5023.6 1345.17  5027.2 1348.09  5035.4 1348.71  5046.4 1350.24  5049.0 1350.99
  5059.8 1354.65  5074.0 1358.70  5092.4 1366.63  5103.1 1372.63  5111.6 1375.69
#Mann=4,-1,0
  4587.3    0.08       0  4995.4    0.05       0  5004.6    0.08       0
  5049.0    0.14       0
#XS Ineff=2,0
    0.00 4930.00 1350.00               0
Permanent Ineff=
       F       F
Bank Sta=4995.4,5004.6
XS Rating Curve= 0
Exp/Cntr=0.3,0.1

Type RM Length L Ch R = 1,75896,290,290,290
BEGIN DESCRIPTION:
South Fork 253.0
END DESCRIPTION:
XS GIS Cut Line= 4
      1431668.05       961451.00      1431445.85       961284.35
      1431386.68       961241.15      1431329.56       961218.39
#Sta/Elev= 30
  4714.5 1361.05  4731.4 1358.17  4751.9 1355.44  4773.3 1353.53  4800.7 1350.46
  4835.2 1347.75  4854.8 1347.02  4866.2 1346.16  4887.2 1345.19  4927.2 1344.25
  4958.0 1344.60  4972.5 1345.22  4979.1 1346.15  4982.5 1345.70  4991.4 1342.07
  4993.2 1340.96  4993.9 1340.89  4995.4 1337.84  4996.9 1334.84  5003.1 1334.84
  5004.6 1337.84  5009.4 1342.16  5013.4 1345.30  5025.9 1347.21  5051.7 1347.40
  5064.4 1348.23  5088.4 1355.37  5102.9 1359.30  5115.8 1365.37  5127.0 1370.04
#Mann=3,-1,0
  4714.5    0.08       0  4995.4    0.05       0  5004.6    0.14       0
#XS Ineff=2,0
    0.00 4900.00 1361.00               0
Permanent Ineff=
       F       F
Bank Sta=4995.4,5004.6
XS Rating Curve= 0
Exp/Cntr=0.3,0.1

Type RM Length L Ch R = 1,75606,269,269,269
BEGIN DESCRIPTION:
South Fork 252.0
END DESCRIPTION:
XS GIS Cut Line= 4
      1431740.98       961161.09      1431685.43       961133.31
      1431490.99       961013.52      1431388.51       961018.73
#Sta/Elev= 30
  4931.9 1363.12  4936.9 1362.05  4942.3 1360.47  4949.6 1356.74  4954.7 1354.56
  4971.2 1345.11  4974.7 1342.51  4992.7 1335.27  4994.0 1335.02  4995.4 1334.31
  4996.9 1331.31  5003.1 1331.31  5004.6 1334.31  5017.1 1338.96  5031.0 1340.73
  5035.7 1340.53  5075.2 1340.75  5084.9 1341.10  5145.9 1342.25  5160.9 1342.17
  5170.3 1342.42  5181.4 1342.09  5202.0 1342.83  5212.6 1343.78  5221.0 1345.04
  5239.6 1346.32  5272.9 1350.80  5299.0 1353.82  5313.5 1356.99  5325.0 1359.89
#Mann=4,-1,0
  4931.9    0.08       0  4995.4    0.05       0  5004.6    0.08       0
  5212.6    0.14       0
Bank Sta=4995.4,5004.6
XS Rating Curve= 0
Exp/Cntr=0.3,0.1

Type RM Length L Ch R = 1,75337,300,300,300
BEGIN DESCRIPTION:
South Fork 251.0
END DESCRIPTION:
XS GIS Cut Line= 4
      1431876.45       960914.57      1431758.38       960881.56
      1431404.18       960813.87      1431339.97       960827.75
#Sta/Elev= 30
  4877.4 1358.91  4902.4 1351.33  4908.8 1349.05  4939.5 1339.24  4944.4 1337.42
  4958.9 1336.35  4969.2 1336.65  4983.9 1333.38  4995.4 1330.81  4996.9 1327.81
  5003.1 1327.81  5004.6 1330.81  5011.8 1338.71  5022.6 1338.26  5045.0 1338.42
  5068.6 1338.25  5103.6 1337.79  5113.9 1337.87  5125.4 1337.49  5174.8 1337.66
  5209.6 1337.51  5260.7 1337.90  5292.4 1338.44  5326.1 1340.30  5369.7 1342.35
  5373.6 1342.86  5388.7 1346.80  5400.7 1349.26  5417.7 1355.51  5426.3 1358.53
#Mann=5,-1,0
  4877.4    0.14       0  4983.9    0.08       0  4995.4    0.05       0
  5004.6    0.08       0  5417.7    0.15       0
#XS Ineff=2,0
       0                 5092.00    0.00 1340.00
Permanent Ineff=
       F       F
Bank Sta=4995.4,5004.6
XS Rating Curve= 0
Exp/Cntr=0.3,0.1

Type RM Length L Ch R = 1,75037,444,444,444
BEGIN DESCRIPTION:
South Fork 250.0
END DESCRIPTION:
XS GIS Cut Line= 3
      1431937.19       960617.69      1431782.40       960619.21
      1431268.73       960589.91
#Sta/Elev= 30
  4845.2 1358.63  4851.9 1358.43  4868.6 1356.56  4880.7 1354.12  4924.2 1342.13
  4937.3 1337.21  4947.9 1335.69  4972.0 1334.57  4981.5 1331.23  4995.4 1327.73
  4996.9 1324.73  5003.1 1324.73  5004.6 1327.73  5005.2 1330.16  5010.1 1332.66
  5115.8 1333.73  5171.0 1333.49  5189.3 1333.84  5213.3 1335.28  5229.1 1334.72
  5260.7 1335.72  5310.8 1335.64  5401.7 1338.71  5423.7 1341.04  5432.7 1342.66
  5450.7 1348.62  5459.2 1351.95  5470.2 1354.36  5479.9 1355.77  5514.5 1365.42
#Mann=5,-1,0
  4845.2    0.14       0  4995.4    0.05       0  5004.6    0.14       0
  5310.8    0.08       0  5450.7    0.15       0
#XS Ineff=2,0
       0                 5150.00    0.00 1336.00
Permanent Ineff=
       F       F
Bank Sta=4995.4,5004.6
XS Rating Curve= 0
Exp/Cntr=0.5,0.3

Type RM Length L Ch R = 1,74593,87,87,87
BEGIN DESCRIPTION:
Haystack Rd US
END DESCRIPTION:
XS GIS Cut Line= 4
      1432062.17       960436.07      1431693.36       960268.92
      1431473.77       960210.13      1431398.62       960209.11
#Sta/Elev= 30
  4525.0 1361.44  4549.7 1357.98  4581.8 1345.97  4593.2 1343.85  4614.6 1342.92
  4625.2 1344.85  4634.2 1344.55  4657.2 1343.97  4694.8 1340.70  4746.6 1332.94
  4756.5 1333.68  4764.6 1332.28  4932.9 1328.88  4964.0 1329.53  4971.4 1330.48
  4990.0 1325.70  4994.0 1321.00  5006.0 1321.00  5010.0 1323.07  5018.9 1324.10
  5027.9 1329.48  5087.3 1331.78  5110.5 1332.13  5120.2 1331.53  5151.9 1335.02
  5159.0 1337.36  5174.0 1338.85  5186.0 1344.30  5207.8 1349.75  5232.4 1357.02
#Mann=4,-1,0
  4525.0    0.14       0  4634.2    0.08       0  4990.0    0.05       0
  5010.0    0.08       0
#XS Ineff=2,0
    0.00 4936.50 1334.10 5063.50    0.00 1336.16
Permanent Ineff=
       F       F
Bank Sta=4990,5010
XS Rating Curve= 0
Exp/Cntr=0.5,0.3

Type RM Length L Ch R =3,74544,,,
BEGIN DESCRIPTION:
Haystack Rd TOR
Structure ID: LDS_SFMR_07
Approximate Survey Structure
END DESCRIPTION:
Bridge Culvert--1,0,-1,-1,0
Deck Dist Width WeirC Skew NumUp NumDn MinLoCord MaxHiCord MaxSubmerge Is_Ogee
33.5,31,3,,26,26,,,0.95,0,1,1,,,
  4485.1  4487.5  4493.1  4498.4  4507.9  4510.6  4571.8  4678.2  4776.1  4899.4
  4970.0  4970.0  5030.0  5030.0  5110.7  5163.7  5165.0  5173.4  5177.5  5185.8
  5191.8  5202.1  5208.1  5213.6  5225.3  5232.3
 1360.16 1359.67 1358.80 1358.03 1359.90 1360.73 1344.32 1339.37 1335.54 1334.23
 1335.20 1335.20 1335.20 1335.20 1338.19 1339.46 1339.60 1340.27 1342.31 1345.50
 1346.99 1349.82 1351.89 1353.44 1356.01 1357.63
 1301.00 1301.00 1301.00 1301.00 1301.00 1301.00 1301.00 1301.00 1301.00 1301.00
 1301.00 1333.00 1333.00 1301.00 1301.00 1301.00 1301.00 1301.00 1301.00 1301.00
 1301.00 1301.00 1301.00 1301.00 1301.00 1301.00
  4485.1  4487.5  4493.1  4498.4  4507.9  4510.6  4571.8  4678.2  4776.1  4899.4
  4970.0  4970.0  5030.0  5030.0  5110.7  5163.7  5165.0  5173.4  5177.5  5185.8
  5191.8  5202.1  5208.1  5213.6  5225.3  5232.3
 1360.16 1359.67 1358.80 1358.03 1359.90 1360.73 1344.32 1339.37 1335.54 1334.23
 1335.20 1335.20 1335.20 1335.20 1338.19 1339.46 1339.60 1340.27 1342.31 1345.50
 1346.99 1349.82 1351.89 1353.44 1356.01 1357.63
 1301.00 1301.00 1301.00 1301.00 1301.00 1301.00 1301.00 1301.00 1301.00 1301.00
 1301.00 1333.00 1333.00 1301.00 1301.00 1301.00 1301.00 1301.00 1301.00 1301.00
 1301.00 1301.00 1301.00 1301.00 1301.00 1301.00
Pier Skew, UpSta & Num, DnSta & Num=,5000,2,5000,2,0,0,0,0,0
       1       1
 1320.00 1333.00
       1       1
 1320.00 1333.00
Abutment Skew #Up #Dn=,2,2
  4970.0  4971.0
 1333.00 1330.43
  4970.0  4971.0
 1333.00 1326.22
Abutment Skew #Up #Dn=,2,2
  5029.0  5030.0
 1329.54 1333.00
  5029.0  5030.0
 1329.52 1333.00
BR Coef=1,1,0,1.25,0,,,0.8,0,2,0,
WSPro=,,,, 1 ,,,, 0 ,,,, 0 ,,,,-1 ,-1 ,-1 , 0 , 0 , 0 , 0 , 0
BC Design=,,0,,0,,,,,,

Type RM Length L Ch R = 1,74506,115,115,115
BEGIN DESCRIPTION:
Haystack Rd DS
END DESCRIPTION:
XS GIS Cut Line= 3
      1432080.50       960331.96      1431482.88       960120.48
      1431400.77       960129.12
#Sta/Elev= 30
  4508.8 1360.90  4526.0 1358.38  4570.2 1348.97  4582.1 1343.84  4592.4 1338.15
  4607.7 1336.48  4613.5 1334.88  4682.5 1331.37  4773.6 1329.32  4784.6 1329.86
  4795.3 1329.12  4902.1 1328.06  4953.3 1328.74  4965.0 1326.85  4976.7 1326.03
  4990.0 1325.50  4994.0 1320.80  5006.0 1320.80  5010.0 1322.25  5018.6 1323.97
  5025.3 1329.17  5034.1 1330.00  5069.2 1330.61  5077.0 1332.22  5097.4 1333.41
  5114.2 1338.35  5175.0 1341.95  5185.4 1343.23  5201.7 1350.28  5225.3 1355.42
#Mann=4,-1,0
  4508.8    0.08       0  4976.7    0.08       0  4990.0    0.05       0
  5010.0    0.08       0
#XS Ineff=2,0
    0.00 4947.50 1334.11 5052.50    0.00 1335.82
Permanent Ineff=
       F       F
Bank Sta=4990,5010
XS Rating Curve= 0
Exp/Cntr=0.5,0.3

Type RM Length L Ch R = 1,74391,254,254,254
BEGIN DESCRIPTION:
South Fork 248.0
END DESCRIPTION:
XS GIS Cut Line= 3
      1432157.49       960055.78      1431618.94       960053.25
      1431407.03       960060.82
#Sta/Elev= 30
  4465.2 1361.89  4510.6 1346.52  4554.3 1333.46  4584.1 1329.91  4617.4 1328.51
  4657.3 1328.44  4675.2 1327.31  4692.4 1327.47  4724.4 1326.62  4954.4 1326.18
  4983.9 1326.54  4988.1 1324.66  4995.4 1321.40  4996.9 1318.40  5003.1 1318.40
  5004.6 1320.00  5020.4 1321.48  5031.5 1321.45  5037.4 1325.80  5057.0 1327.16
  5092.2 1327.69  5096.7 1328.89  5103.4 1329.66  5138.1 1340.19  5144.7 1341.06
  5152.3 1342.89  5196.4 1346.41  5202.8 1348.30  5207.3 1348.66  5215.8 1353.27
#Mann=4,-1,0
  4465.2    0.08       0  4988.1    0.08       0  4995.4    0.05       0
  5004.6    0.08       0
#XS Ineff=2,0
    0.00 4900.00 1328.50               0
Permanent Ineff=
       F       F
Bank Sta=4995.4,5004.6
XS Rating Curve= 0
Exp/Cntr=0.3,0.1

Type RM Length L Ch R = 1,74137,267,267,267
BEGIN DESCRIPTION:
South Fork 247.0
END DESCRIPTION:
XS GIS Cut Line= 3
      1432166.69       959875.79      1431522.12       959847.33
      1431421.92       959841.07
#Sta/Elev= 30
  4354.8 1357.12  4381.1 1351.71  4391.9 1350.05  4401.2 1348.11  4457.3 1334.38
  4484.6 1328.80  4500.2 1326.52  4532.1 1324.61  4580.5 1324.79  4617.2 1324.07
  4658.2 1325.00  4697.7 1324.43  4851.7 1323.88  4928.1 1322.49  4962.1 1323.00
  4964.1 1322.66  4989.4 1318.32  4994.0 1317.90  4996.0 1315.76  5004.0 1315.76
  5006.0 1317.90  5009.9 1318.42  5025.5 1322.84  5034.1 1323.52  5039.0 1323.50
  5050.4 1322.54  5061.8 1323.11  5084.5 1334.95  5095.8 1347.11  5100.4 1349.86
#Mann=4,-1,0
  4354.8    0.08       0  4964.1    0.08       0  4994.0    0.05       0
  5006.0    0.08       0
Bank Sta=4994,5006
XS Rating Curve= 0
Exp/Cntr=0.3,0.1

Type RM Length L Ch R = 1,73870,387,387,387
BEGIN DESCRIPTION:
South Fork 246.0
END DESCRIPTION:
XS GIS Cut Line= 5
      1432223.98       959637.94      1432137.17       959610.28
      1432126.49       959609.69      1431623.28       959613.64
      1431463.53       959615.37
#Sta/Elev= 30
  4376.4 1340.80  4384.7 1338.29  4435.9 1325.75  4447.6 1323.92  4457.2 1322.86
  4479.9 1321.26  4535.8 1320.66  4554.1 1320.17  4578.5 1320.22  4615.9 1320.85
  4756.6 1320.22  4828.2 1320.84  4874.0 1320.89  4921.3 1319.84  4971.9 1319.71
  4979.0 1319.64  4989.7 1318.98  4993.6 1315.05  4995.7 1312.05  5004.3 1312.05
  5006.4 1315.05  5015.9 1317.52  5031.0 1319.12  5058.4 1320.27  5064.4 1319.99
  5077.6 1320.36  5115.6 1325.69  5120.7 1329.26  5127.8 1334.94  5141.2 1345.97
#Mann=5,-1,0
  4376.4    0.08       0  4971.9    0.08       0  4993.6    0.05       0
  5006.4    0.08       0  5127.8     0.1       0
#XS Ineff=2,0
    0.00 4874.00 1324.49               0
Permanent Ineff=
       F       F
Bank Sta=4993.6,5006.4
XS Rating Curve= 0
Exp/Cntr=0.3,0.1

Type RM Length L Ch R = 1,73483,308,308,308
BEGIN DESCRIPTION:
South Fork 245.0
END DESCRIPTION:
XS GIS Cut Line= 4
      1432315.99       959528.57      1431899.32       959299.40
      1431763.91       959288.98      1431644.11       959278.57
#Sta/Elev= 30
  4389.7 1338.28  4397.4 1336.95  4447.4 1326.45  4468.3 1322.83  4509.7 1320.31
  4557.5 1318.69  4592.5 1317.07  4633.8 1316.38  4645.1 1316.91  4713.2 1317.13
  4753.8 1316.80  4835.6 1315.41  4867.5 1313.48  4909.8 1314.81  4928.8 1314.46
  4954.2 1313.32  4977.6 1314.20  4986.1 1312.96  4992.7 1311.31  4995.4 1310.25
  4996.9 1307.25  5003.1 1307.25  5004.6 1310.25  5024.4 1313.91  5039.7 1317.64
  5069.5 1328.68  5074.6 1330.02  5087.2 1331.22  5108.5 1332.01  5121.3 1332.07
#Mann=4,-1,0
  4389.7    0.08       0  4986.1    0.08       0  4995.4    0.05       0
  5004.6    0.08       0
Bank Sta=4995.4,5004.6
XS Rating Curve= 0
Exp/Cntr=0.3,0.1

Type RM Length L Ch R = 1,73175,281,281,281
BEGIN DESCRIPTION:
South Fork 244.0
END DESCRIPTION:
XS GIS Cut Line= 3
      1432451.45       959374.08      1431842.03       959011.21
      1431677.14       958907.06
#Sta/Elev= 30
  4251.2 1335.70  4279.6 1331.12  4313.6 1324.79  4333.9 1322.69  4342.9 1322.44
  4355.2 1319.80  4363.7 1319.14  4479.9 1316.64  4517.8 1316.26  4588.4 1313.61
  4601.4 1313.91  4648.2 1312.69  4808.7 1312.36  4912.1 1311.45  4962.3 1310.35
  4969.4 1309.61  4986.6 1305.59  4990.0 1305.55  4994.1 1305.50  4995.6 1303.56
  5004.4 1303.56  5005.9 1305.50  5017.2 1308.99  5032.6 1311.30  5049.0 1310.83
  5064.4 1311.75  5079.2 1311.65  5091.7 1311.52  5147.7 1332.90  5155.5 1334.89
#Mann=7,-1,0
  4251.2    0.08       0  4279.6    0.08       0  4912.1    0.08       0
  4990.0     0.1       0  4994.1    0.05       0  5005.9     0.1       0
  5079.2    0.08       0
#XS Ineff=2,0
    0.00 4800.00 1314.00               0
Permanent Ineff=
       F       F
Bank Sta=4994.1,5005.9
XS Rating Curve= 0
Exp/Cntr=0.3,0.1

Type RM Length L Ch R = 1,72894,280,280,280
BEGIN DESCRIPTION:
South Fork 243.0
END DESCRIPTION:
XS GIS Cut Line= 4
      1432459.40       959321.96      1432273.75       959223.24
      1431942.91       958839.89      1431906.68       958781.92
#Sta/Elev= 30
  4254.5 1333.03  4268.7 1330.53  4288.9 1326.60  4296.3 1325.55  4300.7 1324.69
  4315.6 1322.07  4338.1 1319.18  4358.6 1317.67  4382.3 1316.77  4409.3 1316.49
  4424.9 1316.76  4463.0 1315.67  4526.5 1314.38  4597.6 1311.83  4613.6 1311.71
  4618.8 1311.28  4625.3 1311.08  4674.2 1310.40  4800.3 1310.66  4900.2 1309.67
  4933.6 1309.44  4975.6 1308.40  4991.0 1307.28  4991.7 1305.32  4993.8 1302.32
  5006.2 1302.32  5008.3 1304.96  5010.6 1304.96  5028.5 1318.12  5039.5 1327.34
#Mann=5,-1,0
  4254.5    0.08       0  4300.7    0.08       0  4900.2    0.08       0
  4991.7    0.05       0  5008.3    0.08       0
#XS Ineff=2,0
    0.00 4766.00 1315.00               0
Permanent Ineff=
       F       F
Bank Sta=4991.7,5008.3
XS Rating Curve= 0
Exp/Cntr=0.3,0.1

Type RM Length L Ch R = 1,72614,319,319,319
BEGIN DESCRIPTION:
South Fork 242.0
END DESCRIPTION:
XS GIS Cut Line= 4
      1432490.22       959291.15      1432368.77       959208.48
      1432198.45       958749.27      1432165.83       958660.47
#Sta/Elev= 30
  4343.6 1331.97  4395.6 1321.16  4421.6 1318.08  4437.3 1316.42  4457.7 1316.35
  4509.8 1314.57  4617.5 1311.87  4662.2 1310.01  4734.0 1307.88  4759.2 1307.74
  4784.6 1306.59  4795.2 1307.23  4830.8 1306.59  4863.6 1306.62  4911.2 1307.70
  4923.8 1307.71  4949.5 1307.13  4965.1 1307.13  4973.4 1307.69  4979.7 1305.79
  4994.1 1301.68  4995.6 1298.68  5004.4 1298.68  5005.9 1301.68  5010.3 1303.96
  5031.8 1305.82  5043.6 1309.57  5058.6 1312.75  5063.1 1315.72  5074.9 1319.84
#Mann=5,-1,0
  4343.6    0.08       0  4421.6    0.08       0  4979.7    0.08       0
  4994.1    0.05       0  5005.9    0.08       0
Bank Sta=4994.1,5005.9
XS Rating Curve= 0
Exp/Cntr=0.3,0.1

Type RM Length L Ch R = 1,72295,258,258,258
BEGIN DESCRIPTION:
South Fork 241.0
END DESCRIPTION:
XS GIS Cut Line= 4
      1432587.22       959233.20      1432532.83       959144.81
      1432476.19       958752.89      1432482.99       958655.50
#Sta/Elev= 30
  4501.7 1334.33  4508.0 1333.43  4531.6 1328.91  4570.3 1320.50  4571.7 1320.15
  4578.0 1317.42  4582.8 1315.98  4608.2 1313.08  4626.2 1311.55  4636.1 1310.74
  4668.8 1309.60  4733.2 1308.32  4818.2 1306.11  4850.9 1305.50  4895.1 1305.27
  4943.5 1303.69  4958.3 1303.55  4980.8 1302.18  4982.2 1302.05  4994.1 1297.53
  4995.6 1295.53  5004.4 1295.53  5005.9 1297.53  5008.2 1298.34  5029.0 1302.12
  5040.8 1304.70  5045.0 1305.21  5060.5 1309.28  5082.9 1314.59  5099.1 1316.64
#Mann=5,-1,0
  4501.7    0.08       0  4626.2    0.08       0  4980.8    0.08       0
  4994.1    0.05       0  5005.9    0.08       0
Bank Sta=4994.1,5005.9
XS Rating Curve= 0
Exp/Cntr=0.3,0.1

Type RM Length L Ch R = 1,72037,292,292,292
BEGIN DESCRIPTION:
South Fork 240.0
END DESCRIPTION:
XS GIS Cut Line= 5
      1432704.10       959151.63      1432664.22       959042.87
      1432719.97       958817.50      1432756.74       958655.46
      1432707.70       958553.50
#Sta/Elev= 30
  4652.0 1327.36  4684.8 1322.89  4699.6 1319.98  4723.7 1313.86  4750.5 1309.07
  4789.3 1305.92  4824.4 1304.25  4857.8 1303.95  4893.0 1301.98  4930.5 1300.70
  4948.0 1301.82  4966.5 1301.19  4994.1 1294.90  4995.6 1292.98  5004.4 1292.98
  5005.9 1295.98  5011.0 1296.57  5017.5 1295.98  5033.4 1299.66  5039.6 1300.09
  5105.3 1302.06  5134.8 1301.87  5146.6 1302.67  5163.1 1302.50  5179.4 1303.03
  5190.0 1304.26  5200.0 1304.74  5224.5 1307.65  5249.0 1314.45  5279.3 1321.72
#Mann=3,-1,0
  4652.0     0.1       0  4994.1    0.05       0  5005.9     0.1       0
Bank Sta=4994.1,5005.9
XS Rating Curve= 0
Exp/Cntr=0.3,0.1

Type RM Length L Ch R = 1,71745,347,347,347
BEGIN DESCRIPTION:
South Fork 239.0
END DESCRIPTION:
XS GIS Cut Line= 3
      1432993.84       959144.23      1432991.01       958920.54
      1432957.03       958328.72
#Sta/Elev= 30
  4769.4 1318.29  4827.3 1315.90  4835.4 1313.94  4868.2 1302.02  4887.3 1298.25
  4899.1 1297.85  4945.5 1298.08  4963.6 1295.73  4993.1 1295.17  4994.1 1292.13
  4995.6 1289.13  5004.4 1289.13  5005.9 1292.13  5008.6 1294.11  5035.2 1296.65
  5070.7 1296.33  5096.8 1297.76  5111.2 1297.50  5132.1 1298.40  5145.4 1297.13
  5157.4 1299.13  5175.7 1299.75  5283.0 1299.08  5333.0 1300.20  5359.6 1301.36
  5386.0 1303.44  5454.3 1305.54  5500.9 1309.11  5541.6 1314.26  5585.9 1323.07
#Mann=3,-1,0
  4769.4     0.1       0  4994.1    0.05       0  5005.9     0.1       0
Bank Sta=4994.1,5005.9
XS Rating Curve= 0
Exp/Cntr=0.3,0.1
