HEC-RAS study South Fork.prj: South Fork Limited Detail Study

--- South Fork.g01 (geometry) --- (continued)

Type RM Length L Ch R = 1,54428,445,445,445
BEGIN DESCRIPTION:
South Fork 181.0
END DESCRIPTION:
XS GIS Cut Line= 3
      1444112.76       958999.62      1443454.40       958427.40
      1443355.99       958349.49
#Sta/Elev= 30
  4411.4 1214.81  4488.5 1211.70  4519.7 1207.47  4583.9 1196.61  4640.8 1192.27
  4775.1 1189.00  4868.6 1188.37  4941.9 1189.04  4977.5 1189.10  4980.7 1187.97
  4984.0 1182.60  4992.7 1180.56  5007.3 1180.56  5008.5 1182.60  5010.9 1185.04
  5019.0 1186.14  5038.4 1186.63  5050.3 1188.55  5074.2 1190.05  5092.9 1189.59
  5224.3 1190.20  5249.1 1189.62  5271.5 1188.97  5323.2 1191.18  5351.8 1190.79
  5366.4 1193.18  5380.2 1193.49  5382.2 1193.86  5405.1 1207.54  5409.2 1210.76
#Mann=6,-1,0
  4411.4    0.08       0  4941.9    0.15       0  4984.0    0.05       0
  5008.5    0.15       0  5092.9    0.08       0  5249.1    0.15       0
#XS Ineff=2,0
    0.00 4700.00 1195.00 5300.00    0.00 1195.00
Permanent Ineff=
       F       F
Bank Sta=4984,5008.5
XS Rating Curve= 0
Exp/Cntr=0.3,0.1

Type RM Length L Ch R = 1,53983,457,457,457
BEGIN DESCRIPTION:
South Fork 180.0
END DESCRIPTION:
XS GIS Cut Line= 3
      1444106.60       958968.82      1443926.13       958427.40
      1443926.13       958390.51
#Sta/Elev= 30
  4656.0 1214.12  4689.9 1212.63  4719.6 1209.75  4795.0 1195.91  4816.3 1192.79
  4891.5 1188.59  4955.0 1187.86  4976.8 1185.51  4984.0 1183.46  4989.4 1182.98
  4990.9 1179.98  5009.1 1179.98  5020.0 1181.98  5023.8 1182.17  5028.7 1184.10
  5042.2 1186.52  5053.5 1186.12  5096.0 1187.61  5121.5 1186.57  5137.6 1187.04
  5142.2 1187.92  5170.3 1188.19  5190.7 1187.04  5220.8 1188.00  5224.4 1189.23
  5233.9 1200.50  5244.8 1203.12  5254.9 1207.75  5260.3 1214.67  5263.6 1217.75
#Mann=4,-1,0
  4656.0    0.08       0  4976.8    0.15       0  4989.4    0.05       0
  5020.0    0.15       0
Bank Sta=4989.4,5020
XS Rating Curve= 0
Exp/Cntr=0.3,0.1

Type RM Length L Ch R = 1,53526,363,363,363
BEGIN DESCRIPTION:
South Fork 179.0
END DESCRIPTION:
XS GIS Cut Line= 3
      1444479.91       958704.30      1444352.73       958546.36
      1444217.36       958388.41
#Sta/Elev= 30
  4690.6 1207.58  4703.2 1205.85  4710.8 1206.05  4713.1 1206.42  4743.4 1204.63
  4750.4 1204.08  4759.3 1202.79  4769.7 1203.50  4800.6 1199.26  4826.9 1196.95
  4831.6 1196.90  4876.0 1192.19  4913.5 1190.56  4930.4 1188.97  4939.5 1188.87
  4953.9 1186.69  4974.5 1182.78  4989.4 1180.62  4990.9 1178.62  5009.1 1178.62
  5020.0 1180.64  5021.4 1180.71  5023.0 1182.61  5028.3 1186.98  5032.9 1187.23
  5047.2 1186.05  5054.2 1186.09  5062.9 1188.78  5071.4 1192.73  5101.4 1211.90
#Mann=3,-1,0
  4690.6    0.15       0  4989.4    0.05       0  5020.0    0.15       0
Bank Sta=4989.4,5020
XS Rating Curve= 0
Exp/Cntr=0.3,0.1

Type RM Length L Ch R = 1,53163,351,351,351
BEGIN DESCRIPTION:
South Fork 177.0
END DESCRIPTION:
XS GIS Cut Line= 3
      1444726.01       958402.78      1444543.48       958226.40
      1444457.34       958130.01
#Sta/Elev= 30
  4683.6 1212.59  4709.9 1209.72  4746.4 1203.86  4766.5 1199.39  4802.9 1191.96
  4808.4 1191.12  4845.0 1188.13  4863.3 1187.60  4890.3 1186.26  4900.9 1185.05
  4905.8 1184.90  4914.9 1183.75  4921.7 1184.71  4940.5 1184.69  4953.0 1185.17
  4972.3 1184.86  4977.5 1183.33  4979.0 1183.17  4986.1 1179.97  4986.8 1179.43
  4987.3 1179.41  4989.1 1177.41  5010.9 1177.41  5012.7 1179.41  5018.4 1179.47
  5024.2 1185.31  5029.9 1192.48  5040.0 1195.59  5048.9 1199.51  5066.7 1209.05
#Mann=3,-1,0
  4683.6    0.15       0  4987.3    0.05       0  5012.7    0.15       0
#XS Ineff=2,0
    0.00 4863.00 1195.00               0
Permanent Ineff=
       F       F
Bank Sta=4987.3,5012.7
XS Rating Curve= 0
Exp/Cntr=0.3,0.1

Type RM Length L Ch R = 1,52812,388,388,388
BEGIN DESCRIPTION:
South Fork 176.0
END DESCRIPTION:
XS GIS Cut Line= 3
      1445052.11       958226.39      1444793.70       957998.74
      1444693.23       957902.37
#Sta/Elev= 30
  4644.0 1213.11  4652.4 1212.68  4672.6 1212.99  4728.9 1207.87  4788.0 1201.83
  4831.4 1195.70  4840.4 1194.39  4860.4 1191.62  4885.1 1189.08  4921.3 1186.93
  4937.9 1185.21  4960.9 1184.81  4968.7 1181.65  4977.7 1180.16  4979.1 1178.99
  4984.1 1178.49  4986.4 1176.49  5013.7 1176.49  5015.9 1178.49  5016.6 1178.49
  5017.6 1180.57  5017.9 1181.75  5031.2 1184.60  5050.1 1184.30  5075.3 1185.20
  5088.9 1189.32  5108.0 1200.66  5113.8 1205.77  5124.9 1210.11  5127.6 1211.64
#Mann=6,-1,0
  4644.0     0.1       0  4831.4    0.15       0  4840.4     0.1       0
  4921.3    0.15       0  4984.1    0.05       0  5015.9    0.15       0
Bank Sta=4984.1,5015.9
XS Rating Curve= 0
Exp/Cntr=0.3,0.1

Type RM Length L Ch R = 1,52424,354,354,354
BEGIN DESCRIPTION:
South Fork 175.0
END DESCRIPTION:
XS GIS Cut Line= 4
      1445417.19       958025.39      1444982.39       957701.35
      1444913.20       957652.19      1444816.26       957615.20
#Sta/Elev= 30
  4444.3 1208.85  4468.9 1207.95  4492.3 1204.47  4511.0 1203.10  4529.6 1200.90
  4581.1 1197.80  4599.9 1196.05  4638.5 1194.22  4676.2 1191.71  4774.9 1186.94
  4885.8 1184.45  4910.8 1184.55  4924.5 1185.19  4949.8 1182.19  4963.0 1182.37
  4968.8 1183.03  4975.2 1177.53  4984.1 1177.07  4986.4 1175.07  5013.7 1175.07
  5015.9 1177.07  5026.8 1183.15  5040.1 1185.32  5044.6 1185.41  5064.6 1188.76
  5079.6 1190.57  5093.2 1191.27  5123.8 1196.21  5160.5 1200.78  5175.2 1202.07
#Mann=4,-1,0
  4444.3    0.08       0  4885.8    0.15       0  4984.1    0.05       0
  5015.9    0.15       0
Bank Sta=4984.1,5015.9
XS Rating Curve= 0
Exp/Cntr=0.3,0.1

Type RM Length L Ch R = 1,52070,278,278,278
BEGIN DESCRIPTION:
South Fork 174.0
END DESCRIPTION:
XS GIS Cut Line= 3
      1445550.50       957916.68      1445230.56       957471.63
      1445134.17       957352.69
#Sta/Elev= 30
  4398.2 1207.67  4423.5 1204.76  4436.7 1202.27  4446.6 1201.35  4479.1 1200.27
  4496.9 1198.46  4534.3 1195.83  4572.4 1190.87  4623.7 1186.98  4724.0 1183.19
  4794.1 1182.19  4813.2 1182.76  4845.5 1182.40  4894.7 1183.78  4914.3 1181.69
  4947.5 1181.80  4972.1 1180.05  4973.9 1177.03  4977.7 1176.72  4980.9 1174.72
  5019.1 1174.72  5022.3 1176.72  5024.9 1177.73  5042.3 1181.78  5050.7 1182.63
  5061.0 1184.39  5065.5 1187.70  5079.9 1195.60  5087.9 1202.71  5099.4 1208.55
#Mann=4,-1,0
  4398.2    0.08       0  4845.5    0.15       0  4977.7    0.05       0
  5022.3    0.15       0
#XS Ineff=2,0
    0.00 4700.00 1187.00               0
Permanent Ineff=
       F       F
Bank Sta=4977.7,5022.3
XS Rating Curve= 0
Exp/Cntr=0.5,0.3

Type RM Length L Ch R = 1,51792,79,79,79
BEGIN DESCRIPTION:
Zephyr Mountain Park Rd US
END DESCRIPTION:
XS GIS Cut Line= 5
      1445638.70       957828.49      1445517.70       957559.83
      1445443.13       957312.27      1445426.23       957256.27
      1445393.66       957226.23
#Sta/Elev= 30
  4467.3 1202.96  4524.1 1197.87  4529.4 1198.82  4566.3 1190.09  4587.4 1189.53
  4603.2 1191.50  4647.3 1191.94  4679.7 1190.79  4733.5 1185.31  4759.1 1185.86
  4766.1 1181.91  4803.4 1182.86  4814.5 1180.83  4857.2 1180.97  4918.4 1181.51
  4955.7 1177.49  4969.7 1178.74  4980.0 1176.48  4987.5 1172.80  5012.5 1172.80
  5020.0 1176.48  5025.1 1176.51  5026.0 1178.20  5031.9 1179.72  5035.4 1182.30
  5040.2 1183.07  5054.7 1181.48  5083.7 1181.94  5102.6 1197.09  5123.3 1203.16
#Mann=4,-1,0
  4467.3    0.08       0  4857.2    0.15       0  4980.0    0.05       0
  5020.0    0.15       0
#XS Ineff=2,0
    0.00 4936.80 1186.00 5063.30    0.00 1186.24
Permanent Ineff=
       F       F
Bank Sta=4980,5020
XS Rating Curve= 0
Exp/Cntr=0.5,0.3

Type RM Length L Ch R =3,51754,,,
BEGIN DESCRIPTION:
Zephyr Mountain Park Rd TOR
Structure ID: LDS_SFMR_05
Approximate Survey Structure
END DESCRIPTION:
Bridge Culvert--1,0,-1,-1,0
Deck Dist Width WeirC Skew NumUp NumDn MinLoCord MaxHiCord MaxSubmerge Is_Ogee
23,30,3,,44,44,,,0.95,0,1,1,,,
  4469.5  4477.4  4479.1  4482.0  4495.5  4498.6  4500.7  4513.1  4514.7  4517.1
  4519.5  4522.0  4533.2  4535.7  4538.1  4551.3  4551.6  4551.9  4556.4  4570.3
  4574.4  4575.1  4575.9  4589.1  4590.7  4593.9  4757.8  4830.8  4884.9  4909.1
  4940.8  4953.0  4959.8  4959.8  5040.3  5040.3  5042.5  5089.9  5117.5  5128.5
  5133.7  5149.7  5166.3  5202.0
 1208.13 1207.80 1207.70 1207.44 1206.42 1206.30 1206.17 1205.69 1205.66 1205.41
 1205.13 1205.14 1204.72 1204.39 1204.19 1203.82 1203.79 1203.79 1203.33 1202.61
 1202.04 1201.97 1201.95 1201.38 1201.27 1200.95 1191.05 1188.10 1186.75 1186.52
 1186.16 1186.20 1186.20 1186.20 1186.20 1186.20 1186.20 1186.18 1186.23 1189.70
 1191.44 1198.09 1202.06 1206.18
 1152.80 1152.80 1152.80 1152.80 1152.80 1152.80 1152.80 1152.80 1152.80 1152.80
 1152.80 1152.80 1152.80 1152.80 1152.80 1152.80 1152.80 1152.80 1152.80 1152.80
 1152.80 1152.80 1152.80 1152.80 1152.80 1152.80 1152.80 1152.80 1152.80 1152.80
 1152.80 1152.80 1152.80 1184.20 1184.20 1152.80 1152.80 1152.80 1152.80 1152.80
 1152.80 1152.80 1152.80 1152.80
  4469.5  4477.4  4479.1  4482.0  4495.5  4498.6  4500.7  4513.1  4514.7  4517.1
  4519.5  4522.0  4533.2  4535.7  4538.1  4551.3  4551.6  4551.9  4556.4  4570.3
  4574.4  4575.1  4575.9  4589.1  4590.7  4593.9  4757.8  4830.8  4884.9  4909.1
  4940.8  4953.0  4959.8  4959.8  5040.3  5040.3  5042.5  5089.9  5117.5  5128.5
  5133.7  5149.7  5166.3  5202.0
 1208.13 1207.80 1207.70 1207.44 1206.42 1206.30 1206.17 1205.69 1205.66 1205.41
 1205.13 1205.14 1204.72 1204.39 1204.19 1203.82 1203.79 1203.79 1203.33 1202.61
 1202.04 1201.97 1201.95 1201.38 1201.27 1200.95 1191.05 1188.10 1186.75 1186.52
 1186.16 1186.20 1186.20 1186.20 1186.20 1186.20 1186.20 1186.18 1186.23 1189.70
 1191.44 1198.09 1202.06 1206.18
 1152.80 1152.80 1152.80 1152.80 1152.80 1152.80 1152.80 1152.80 1152.80 1152.80
 1152.80 1152.80 1152.80 1152.80 1152.80 1152.80 1152.80 1152.80 1152.80 1152.80
 1152.80 1152.80 1152.80 1152.80 1152.80 1152.80 1152.80 1152.80 1152.80 1152.80
 1152.80 1152.80 1152.80 1184.20 1184.20 1152.80 1152.80 1152.80 1152.80 1152.80
 1152.80 1152.80 1152.80 1152.80
Pier Skew, UpSta & Num, DnSta & Num=,5000,2,5000,2,0,0,0,0,0
       3       3
 1172.80 1184.20
       3       3
 1172.55 1184.20
Abutment Skew #Up #Dn=,2,2
  4959.8  4974.8
 1184.20 1177.64
  4959.8  4974.9
 1184.20 1179.17
Abutment Skew #Up #Dn=,2,2
  5025.3  5040.3
 1176.89 1184.20
  5025.3  5040.3
 1178.39 1184.20
BR Coef=1,1,0,1.25,0,,,0.8,0,2,0,
WSPro=,,,, 1 ,,,, 0 ,,,, 0 ,,,,-1 ,-1 ,-1 , 0 , 0 , 0 , 0 , 0
BC Design=,,0,,0,,,,,,

Type RM Length L Ch R = 1,51713,536,536,536
BEGIN DESCRIPTION:
Zephyr Mountain Park Rd DS
END DESCRIPTION:
XS GIS Cut Line= 5
      1445720.76       957799.82      1445585.38       957559.83
      1445520.87       957295.77      1445508.44       957236.09
      1445394.52       957194.82
#Sta/Elev= 30
  4472.0 1209.05  4493.3 1207.11  4504.3 1208.41  4564.9 1208.04  4569.2 1209.66
  4588.5 1207.73  4625.0 1207.58  4634.3 1205.30  4660.1 1201.87  4669.7 1201.94
  4698.6 1197.54  4823.1 1185.87  4864.9 1180.91  4908.2 1180.39  4921.6 1178.21
  4951.8 1180.71  4978.7 1178.94  4980.0 1176.41  4987.5 1172.55  5012.5 1172.55
  5020.0 1176.41  5023.4 1176.42  5028.6 1181.28  5080.3 1181.11  5108.9 1184.78
  5138.3 1185.79  5153.8 1188.03  5174.4 1195.30  5195.4 1200.36  5201.5 1200.65
#Mann=4,-1,0
  4472.0    0.08       0  4823.1    0.15       0  4980.0    0.05       0
  5020.0    0.15       0
#XS Ineff=2,0
    0.00 4933.80 1185.88 5066.30    0.00 1186.15
Permanent Ineff=
       F       F
Bank Sta=4980,5020
XS Rating Curve= 0
Exp/Cntr=0.5,0.3

Type RM Length L Ch R = 1,51177,438,438,438
BEGIN DESCRIPTION:
South Fork 171.0
END DESCRIPTION:
XS GIS Cut Line= 4
      1446244.01       956996.53      1446142.48       956952.27
      1445270.17       956891.21      1445137.30       956819.47
#Sta/Elev= 30
  4299.8 1226.29  4407.2 1211.55  4473.8 1191.36  4496.3 1187.11  4530.0 1185.06
  4571.4 1185.05  4674.0 1181.23  4813.8 1181.16  4835.8 1181.79  4964.6 1177.24
  4974.4 1179.02  4978.4 1175.72  4986.2 1174.61  4988.2 1171.61  5011.8 1171.61
  5013.8 1174.61  5029.6 1175.72  5040.4 1179.79  5134.7 1181.23  5149.3 1187.92
  5157.3 1188.09  5186.2 1188.10  5198.3 1182.57  5207.1 1181.53  5285.0 1178.89
  5333.5 1178.53  5374.2 1186.58  5394.8 1192.11  5416.0 1193.86  5436.0 1203.99
#Mann=4,-1,0
  4299.8    0.08       0  4813.8    0.15       0  4986.2    0.05       0
  5013.8    0.15       0
#XS Ineff=2,0
    0.00 4900.00 1182.00 5157.30    0.00 1190.00
Permanent Ineff=
       F       F
Bank Sta=4986.2,5013.8
XS Rating Curve= 0
Exp/Cntr=0.3,0.1

Type RM Length L Ch R = 1,50739,387,387,387
BEGIN DESCRIPTION:
South Fork 169.0
END DESCRIPTION:
XS GIS Cut Line= 4
      1446301.33       956861.12      1446173.73       956777.79
      1445464.19       956428.69      1445324.79       956408.00
#Sta/Elev= 30
  4190.3 1215.38  4254.9 1202.20  4259.7 1200.15  4293.8 1191.08  4313.8 1187.70
  4333.8 1184.49  4353.7 1182.59  4392.9 1182.70  4411.6 1179.14  4416.9 1180.11
  4511.7 1178.15  4620.0 1178.64  4714.9 1178.07  4817.1 1176.07  4922.4 1176.25
  4959.7 1176.97  4969.5 1176.02  4985.3 1172.08  4987.3 1169.08  5012.7 1169.08
  5035.0 1172.08  5036.5 1172.24  5040.2 1172.63  5042.9 1174.93  5053.5 1176.89
  5079.9 1176.45  5119.6 1177.72  5182.2 1182.50  5211.3 1193.51  5274.4 1209.88
#Mann=5,-1,0
  4190.3    0.08       0  4922.4    0.15       0  4985.3    0.05       0
  5035.0    0.15       0  5036.5    0.08       0
#XS Ineff=2,0
    0.00 4800.00 1185.00               0
Permanent Ineff=
       F       F
Bank Sta=4985.3,5035
XS Rating Curve= 0
Exp/Cntr=0.3,0.1

Type RM Length L Ch R = 1,50352,552,552,552
BEGIN DESCRIPTION:
South Fork 168.0
END DESCRIPTION:
XS GIS Cut Line= 3
      1446604.68       956603.29      1445891.83       956235.47
      1445393.80       956004.36
#Sta/Elev= 30
  4140.2 1220.19  4194.5 1210.01  4215.3 1204.75  4275.1 1194.08  4367.2 1183.24
  4409.5 1180.45  4471.5 1179.17  4477.7 1177.78  4626.5 1176.42  4813.2 1176.75
  4895.2 1174.26  4950.5 1174.25  4972.4 1176.01  4976.2 1176.59  4982.7 1171.99
  4988.7 1169.50  4990.2 1166.50  5009.8 1166.50  5011.3 1169.50  5032.4 1172.00
  5033.0 1173.75  5037.2 1175.33  5048.7 1175.02  5202.5 1174.06  5372.3 1176.86
  5397.5 1180.46  5412.7 1192.10  5437.7 1200.37  5454.9 1203.36  5491.4 1206.40
#Mann=5,-1,0
  4140.2    0.08       0  4972.4    0.15       0  4988.7    0.05       0
  5011.3    0.15       0  5048.7    0.08       0
#XS Ineff=2,0
    0.00 4800.00 1180.00 5250.00    0.00 1179.35
Permanent Ineff=
       F       F
Bank Sta=4988.7,5011.3
XS Rating Curve= 0
Exp/Cntr=0.3,0.1

Type RM Length L Ch R = 1,49800,988,988,988
BEGIN DESCRIPTION:
South Fork 166.0
END DESCRIPTION:
XS GIS Cut Line= 3
      1446660.05       956339.63      1445995.67       955695.60
      1445924.38       955623.49
#Sta/Elev= 30
  4074.7 1198.37  4153.0 1185.54  4179.4 1181.79  4212.9 1178.26  4299.9 1172.41
  4343.1 1171.82  4362.6 1169.37  4379.3 1170.46  4434.9 1171.21  4441.1 1172.29
  4520.4 1171.61  4587.6 1172.91  4713.9 1173.88  4776.9 1171.93  4827.2 1171.76
  4891.4 1172.87  4937.0 1173.08  4957.1 1174.58  4966.5 1167.78  4978.5 1167.34
  4981.4 1164.34  5018.6 1164.34  5021.5 1167.34  5032.8 1171.68  5039.0 1176.87
  5052.8 1184.57  5058.3 1189.67  5071.9 1200.30  5097.5 1217.63  5101.4 1218.61
#Mann=4,-1,0
  4074.7    0.08       0  4891.4    0.15       0  4978.5    0.05       0
  5021.5    0.15       0
#XS Ineff=2,0
    0.00 4600.00 1180.00               0
Permanent Ineff=
       F       F
Bank Sta=4978.5,5021.5
XS Rating Curve= 0
Exp/Cntr=0.3,0.1

Type RM Length L Ch R = 1,48812,640,640,640
BEGIN DESCRIPTION:
South Fork 164.0
END DESCRIPTION:
XS GIS Cut Line= 3
      1446686.08       956284.33      1446993.12       955693.63
      1447063.68       955636.53
#Sta/Elev= 30
  4587.6 1196.14  4614.4 1194.82  4628.9 1190.00  4671.4 1171.33  4677.4 1169.88
  4712.8 1168.07  4821.9 1169.49  4851.0 1168.85  4895.7 1169.66  4943.3 1169.36
  4981.9 1170.23  4984.6 1169.69  4985.5 1166.64  4988.5 1165.20  4990.0 1162.20
  5010.0 1162.20  5011.5 1165.20  5017.0 1165.53  5035.7 1166.63  5036.7 1168.04
  5045.1 1170.45  5060.5 1169.17  5092.3 1169.79  5123.5 1174.37  5155.9 1178.67
  5188.8 1181.00  5204.4 1181.16  5253.3 1185.23  5329.2 1194.75  5344.1 1198.32
#Mann=7,-1,0
  4587.6    0.15       0  4712.8    0.08       0  4943.3    0.15       0
  4988.5    0.05       0  5011.5    0.15       0  5017.0    0.08       0
  5123.5    0.15       0
Bank Sta=4988.5,5011.5
XS Rating Curve= 0
Exp/Cntr=0.3,0.1

Type RM Length L Ch R = 1,48172,520,520,520
BEGIN DESCRIPTION:
South Fork 162.0
END DESCRIPTION:
XS GIS Cut Line= 3
      1446949.76       956443.82      1447327.38       955939.25
      1447382.75       955900.16
#Sta/Elev= 30
  4892.0 1187.18  4897.1 1184.23  4916.4 1174.47  4930.3 1171.35  4944.7 1169.14
  4959.4 1167.65  4960.8 1166.50  4972.5 1166.04  4977.3 1162.19  4978.2 1162.15
  4981.0 1159.15  5019.0 1159.15  5048.1 1162.15  5064.8 1166.39  5067.5 1167.02
  5083.0 1168.27  5141.9 1167.92  5216.0 1168.23  5248.7 1167.71  5356.2 1167.53
  5396.4 1167.93  5445.9 1169.90  5461.7 1171.19  5474.3 1172.94  5487.3 1176.19
  5489.9 1176.50  5506.8 1181.26  5534.7 1186.99  5548.2 1190.81  5590.0 1200.42
#Mann=5,-1,0
  4892.0    0.15       0  4978.2    0.05       0  5048.1    0.15       0
  5064.8    0.08       0  5445.9    0.15       0
#XS Ineff=2,0
       0                 5150.00    0.00 1169.00
Permanent Ineff=
       F       F
Bank Sta=4978.2,5048.1
XS Rating Curve= 0
Exp/Cntr=0.3,0.1

Type RM Length L Ch R = 1,47652,577,577,577
BEGIN DESCRIPTION:
South Fork 159.0
END DESCRIPTION:
XS GIS Cut Line= 3
      1447372.95       956674.92      1447457.58       956570.76
      1447779.85       956199.67
#Sta/Elev= 30
  4833.2 1192.57  4835.0 1192.19  4840.0 1189.15  4847.2 1185.91  4853.9 1181.72
  4859.7 1180.82  4868.2 1176.23  4871.2 1171.75  4882.0 1167.97  4940.3 1164.07
  4956.4 1163.95  4974.5 1160.56  4978.2 1159.12  4981.0 1156.12  5019.0 1156.12
  5021.9 1159.12  5030.5 1159.82  5033.6 1161.03  5035.1 1163.38  5052.1 1165.98
  5066.4 1166.86  5112.1 1165.08  5159.1 1165.99  5175.0 1165.13  5237.7 1164.41
  5273.7 1164.72  5345.5 1165.40  5384.0 1174.50  5412.6 1184.57  5458.9 1198.71
#Mann=5,-1,0
  4833.2    0.15       0  4978.2    0.05       0  5021.9    0.15       0
  5052.1    0.08       0  5273.7    0.15       0
#XS Ineff=2,0
       0                 5200.00    0.00 1169.00
Permanent Ineff=
       F       F
Bank Sta=4978.2,5021.9
XS Rating Curve= 0
Exp/Cntr=0.3,0.1

Type RM Length L Ch R = 1,47075,575,575,575
BEGIN DESCRIPTION:
South Fork 157.0
END DESCRIPTION:
XS GIS Cut Line= 3
      1447568.28       956899.51      1447929.59       956482.87
      1448036.99       956342.92
#Sta/Elev= 30
  4449.2 1190.47  4460.7 1185.50  4476.1 1181.30  4488.7 1175.76  4520.4 1169.61
  4544.0 1167.51  4560.6 1166.54  4575.6 1166.50  4606.3 1167.95  4621.4 1167.80
  4667.0 1166.12  4757.6 1164.90  4898.9 1165.36  4927.5 1165.33  4961.9 1163.90
  4973.4 1158.67  4973.7 1156.92  4974.7 1156.88  4978.0 1153.88  5022.0 1153.88
  5025.3 1156.88  5026.4 1156.88  5028.4 1158.76  5032.3 1169.00  5039.0 1170.13
  5050.7 1177.08  5056.5 1179.13  5084.2 1182.83  5120.6 1187.11  5177.1 1192.28
#Mann=6,-1,0
  4449.2    0.15       0  4544.0    0.08       0  4898.9    0.15       0
  4974.7    0.05       0  5025.3    0.15       0  5084.2    0.08       0
Bank Sta=4974.7,5025.3
XS Rating Curve= 0
Exp/Cntr=0.3,0.1

Type RM Length L Ch R = 1,46500,663,663,663
BEGIN DESCRIPTION:
South Fork 155.0
END DESCRIPTION:
XS GIS Cut Line= 3
      1447903.52       957153.47      1448300.71       956828.65
      1448463.48       956710.71
#Sta/Elev= 30
  4486.9 1188.35  4513.5 1187.45  4524.8 1185.98  4536.7 1186.35  4548.5 1184.62
  4572.9 1182.26  4586.4 1181.87  4602.0 1181.92  4618.0 1181.35  4638.5 1179.12
  4698.5 1175.05  4772.5 1167.62  4796.4 1165.62  4824.8 1164.05  4923.6 1161.99
  4954.2 1161.33  4966.7 1156.26  4967.2 1155.75  4970.1 1155.70  4974.0 1152.70
  5026.0 1152.70  5029.9 1155.70  5030.6 1157.45  5044.8 1161.13  5062.2 1161.83
  5108.6 1164.59  5124.4 1168.16  5168.5 1185.90  5181.3 1190.48  5201.0 1195.99
#Mann=4,-1,0
  4486.9    0.08       0  4923.6    0.15       0  4970.1    0.05       0
  5029.9    0.15       0
Bank Sta=4970.1,5029.9
XS Rating Curve= 0
Exp/Cntr=0.3,0.1

Type RM Length L Ch R = 1,45837,428,428,428
BEGIN DESCRIPTION:
South Fork 153.0
END DESCRIPTION:
XS GIS Cut Line= 3
      1448333.27       957521.25      1448860.58       957114.38
      1448941.92       957052.56
#Sta/Elev= 30
  4340.6 1196.28  4426.1 1181.94  4487.5 1174.37  4524.9 1171.45  4604.8 1168.41
  4724.4 1165.58  4761.8 1162.74  4807.3 1160.90  4838.7 1160.17  4855.3 1160.53
  4870.1 1162.12  4877.6 1162.57  4902.6 1159.66  4916.2 1156.23  4928.2 1157.09
  4940.9 1154.58  4952.5 1155.11  4965.8 1158.05  4975.0 1157.93  4977.8 1157.23
  4978.8 1153.51  4979.3 1153.44  4982.0 1150.44  5018.0 1150.44  5030.1 1153.44
  5032.0 1153.44  5033.5 1158.57  5035.7 1161.05  5063.1 1173.92  5108.8 1186.71
#Mann=4,-1,0
  4340.6    0.08       0  4870.1    0.15       0  4979.3    0.05       0
  5030.1    0.15       0
Bank Sta=4979.3,5030.1
XS Rating Curve= 0
Exp/Cntr=0.3,0.1

Type RM Length L Ch R = 1,45409,505,505,505
BEGIN DESCRIPTION:
South Fork 151.0
END DESCRIPTION:
XS GIS Cut Line= 4
      1448538.33       957719.84      1449062.40       957488.73
      1449283.76       957400.84      1449332.56       957378.06
#Sta/Elev= 30
  4450.4 1196.41  4467.0 1194.95  4497.6 1188.32  4509.1 1186.93  4579.8 1185.29
  4608.6 1183.63  4653.0 1177.48  4738.0 1170.21  4756.9 1167.69  4789.6 1161.38
  4832.7 1156.62  4961.9 1157.05  4967.1 1154.08  4973.9 1153.85  4974.1 1149.01
  4974.7 1149.01  4978.0 1146.01  5022.0 1146.01  5029.0 1149.01  5029.9 1149.01
  5033.2 1156.99  5034.8 1158.67  5051.7 1157.62  5192.5 1155.87  5211.4 1155.56
  5236.5 1157.56  5251.7 1166.75  5264.9 1173.00  5304.6 1186.62  5315.2 1188.96
#Mann=4,-1,0
  4450.4     0.1       0  4974.7    0.05       0  5029.0     0.1       0
  5192.5    0.15       0
#XS Ineff=2,0
    0.00 4950.00 1196.00 5200.00    0.00 1160.00
Permanent Ineff=
       F       F
Bank Sta=4974.7,5029
XS Rating Curve= 0
Exp/Cntr=0.3,0.1

Type RM Length L Ch R = 1,44904,281,281,281
BEGIN DESCRIPTION:
South Fork 149.0
END DESCRIPTION:
XS GIS Cut Line= 5
      1449273.99       958201.65      1449293.52       957892.37
      1449414.65       957681.18      1449420.48       957671.02
      1449495.33       957534.34
#Sta/Elev= 30
  4348.2 1195.54  4433.5 1179.39  4457.5 1176.55  4474.5 1173.26  4492.6 1169.06
  4507.2 1166.91  4536.2 1164.01  4584.1 1161.13  4643.4 1159.53  4658.4 1159.88
  4689.9 1159.48  4704.7 1159.96  4756.4 1159.28  4815.4 1157.27  4880.0 1154.45
  4889.1 1153.62  4904.0 1154.07  4935.3 1153.33  4944.0 1153.47  4960.4 1155.16
  4968.2 1148.75  4977.3 1147.94  4979.7 1144.94  5020.3 1144.94  5022.7 1147.94
  5023.3 1148.08  5026.3 1162.16  5043.7 1167.68  5062.3 1183.68  5069.1 1185.93
#Mann=6,-1,0
  4348.2     0.1       0  4756.4    0.08       0  4815.4     0.1       0
  4880.0    0.15       0  4977.3    0.05       0  5022.7    0.15       0
Bank Sta=4977.3,5022.7
XS Rating Curve= 0
Exp/Cntr=0.5,0.3

Type RM Length L Ch R = 1,44623,58,58,58
BEGIN DESCRIPTION:
Golden Rd US
END DESCRIPTION:
XS GIS Cut Line= 4
      1449456.27       958230.93      1449635.33       957889.21
      1449669.24       957730.95      1449622.31       957612.45
#Sta/Elev= 30
  4510.2 1182.40  4531.6 1179.38  4546.4 1176.52  4576.1 1172.92  4606.1 1170.25
  4634.6 1168.61  4705.8 1166.14  4785.2 1162.05  4826.0 1160.88  4882.9 1157.61
  4886.1 1157.73  4916.1 1155.63  4932.7 1155.26  4950.0 1153.96  4953.9 1154.18
  4962.3 1151.98  4977.5 1152.00  4985.0 1144.70  5015.0 1144.70  5022.5 1152.00
  5053.4 1156.51  5057.8 1156.93  5072.5 1156.30  5091.9 1159.04  5100.8 1159.47
  5122.2 1163.87  5133.4 1165.64  5146.7 1168.47  5158.2 1171.56  5185.3 1175.39
#Mann=4,-1,0
  4510.2    0.08       0  4916.1    0.15       0  4977.5    0.05       0
  5022.5    0.15       0
#XS Ineff=2,0
    0.00 4958.00 1157.30 5042.00    0.00 1157.30
Permanent Ineff=
       F       F
Bank Sta=4977.5,5022.5
XS Rating Curve= 0
Exp/Cntr=0.5,0.3

Type RM Length L Ch R =3,44593,,,
BEGIN DESCRIPTION:
Golden Rd TOR
Structure ID: LDS_SFMR_04
Approximate Survey Structure
END DESCRIPTION:
Bridge Culvert--1,0,-1,-1,0
Deck Dist Width WeirC Skew NumUp NumDn MinLoCord MaxHiCord MaxSubmerge Is_Ogee
17,26,3,,56,56,,,0.95,0,1,1,,,
  4492.9  4493.2  4504.7  4508.3  4529.7  4537.5  4563.6  4575.1  4576.8  4579.2
  4590.8  4599.1  4611.2  4629.9  4635.1  4645.0  4647.5  4663.3  4671.3  4676.4
  4682.6  4695.4  4702.3  4716.7  4717.4  4729.8  4846.4  4909.9  4928.3  4975.0
  4975.0  5025.0  5025.0  5045.4  5072.9  5075.2  5077.5  5088.0  5092.0  5097.9
  5101.0  5115.1  5123.1  5142.5  5159.5  5161.4  5170.9  5171.1  5185.6  5189.5
  5193.7  5204.9  5208.7  5212.4  5217.6  5245.4
 1180.99 1180.95 1180.02 1179.61 1177.53 1177.04 1174.44 1173.46 1173.26 1173.10
 1172.22 1171.42 1170.63 1169.05 1168.72 1168.25 1168.10 1166.72 1166.28 1166.23
 1166.11 1165.35 1164.88 1164.18 1164.17 1163.67 1159.81 1157.81 1157.30 1157.30
 1157.30 1157.30 1157.30 1157.30 1159.61 1159.78 1160.02 1160.66 1160.99 1161.41
 1161.55 1162.78 1163.35 1165.62 1167.95 1168.14 1169.52 1169.57 1171.45 1172.00
 1172.48 1174.16 1174.52 1175.16 1175.73 1178.96
 1124.70 1124.70 1124.70 1124.70 1124.70 1124.70 1124.70 1124.70 1124.70 1124.70
 1124.70 1124.70 1124.70 1124.70 1124.70 1124.70 1124.70 1124.70 1124.70 1124.70
 1124.70 1124.70 1124.70 1124.70 1124.70 1124.70 1124.70 1124.70 1124.70 1124.70
 1154.50 1154.50 1124.70 1124.70 1124.70 1124.70 1124.70 1124.70 1124.70 1124.70
 1124.70 1124.70 1124.70 1124.70 1124.70 1124.70 1124.70 1124.70 1124.70 1124.70
 1124.70 1124.70 1124.70 1124.70 1124.70 1124.70
  4492.9  4493.2  4504.7  4508.3  4529.7  4537.5  4563.6  4575.1  4576.8  4579.2
  4590.8  4599.1  4611.2  4629.9  4635.1  4645.0  4647.5  4663.3  4671.3  4676.4
  4682.6  4695.4  4702.3  4716.7  4717.4  4729.8  4846.4  4909.9  4928.3  4975.0
  4975.0  5025.0  5025.0  5045.4  5072.9  5075.2  5077.5  5088.0  5092.0  5097.9
  5101.0  5115.1  5123.1  5142.5  5159.5  5161.4  5170.9  5171.1  5185.6  5189.5
  5193.7  5204.9  5208.7  5212.4  5217.6  5245.4
 1180.99 1180.95 1180.02 1179.61 1177.53 1177.04 1174.44 1173.46 1173.26 1173.10
 1172.22 1171.42 1170.63 1169.05 1168.72 1168.25 1168.10 1166.72 1166.28 1166.23
 1166.11 1165.35 1164.88 1164.18 1164.17 1163.67 1159.81 1157.81 1157.30 1157.30
 1157.30 1157.30 1157.30 1157.30 1159.61 1159.78 1160.02 1160.66 1160.99 1161.41
 1161.55 1162.78 1163.35 1165.62 1167.95 1168.14 1169.52 1169.57 1171.45 1172.00
 1172.48 1174.16 1174.52 1175.16 1175.73 1178.96
 1124.70 1124.70 1124.70 1124.70 1124.70 1124.70 1124.70 1124.70 1124.70 1124.70
 1124.70 1124.70 1124.70 1124.70 1124.70 1124.70 1124.70 1124.70 1124.70 1124.70
 1124.70 1124.70 1124.70 1124.70 1124.70 1124.70 1124.70 1124.70 1124.70 1124.70
 1154.50 1154.50 1124.70 1124.70 1124.70 1124.70 1124.70 1124.70 1124.70 1124.70
 1124.70 1124.70 1124.70 1124.70 1124.70 1124.70 1124.70 1124.70 1124.70 1124.70
 1124.70 1124.70 1124.70 1124.70 1124.70 1124.70
Abutment Skew #Up #Dn=,2,2
  4975.0  4976.0
 1154.50 1153.98
  4975.0  4976.0
 1154.50 1147.22
Abutment Skew #Up #Dn=,2,2
  5024.0  5025.0
 1153.40 1154.50
  5024.0  5025.0
 1152.79 1154.50
BR Coef=1,1,0,1.25,0,,,0.8,0,2,0,
WSPro=,,,, 1 ,,,, 0 ,,,, 0 ,,,,-1 ,-1 ,-1 , 0 , 0 , 0 , 0 , 0
BC Design=,,0,,0,,,,,,

Type RM Length L Ch R = 1,44565,591,591,591
BEGIN DESCRIPTION:
Golden Rd DS
END DESCRIPTION:
XS GIS Cut Line= 4
      1449658.10       958292.80      1449661.36       958009.56
      1449732.98       957719.85      1449671.13       957576.63
#Sta/Elev= 30
  4509.8 1177.10  4537.0 1172.17  4572.7 1167.46  4595.9 1166.26  4607.6 1166.82
  4643.7 1166.43  4681.8 1163.49  4713.1 1162.07  4730.4 1161.28  4769.6 1161.44
  4875.2 1155.19  4910.8 1154.68  4953.5 1155.71  4956.6 1154.48  4977.5 1151.81
  4985.0 1144.45  5015.0 1144.45  5022.5 1152.00  5033.9 1154.23  5052.4 1154.77
  5090.6 1158.58  5112.0 1159.70  5155.4 1164.35  5172.0 1165.05  5183.4 1164.53
  5192.5 1165.47  5217.4 1169.55  5228.2 1170.43  5231.7 1173.34  5247.5 1176.73
#Mann=5,-1,0
  4509.8    0.15       0  4713.1    0.08       0  4910.8    0.15       0
  4977.5    0.05       0  5022.5    0.15       0
#XS Ineff=2,0
    0.00 4960.00 1157.30 5040.00    0.00 1157.30
Permanent Ineff=
       F       F
Bank Sta=4977.5,5022.5
XS Rating Curve= 0
Exp/Cntr=0.5,0.3

Type RM Length L Ch R = 1,43974,522,522,522
BEGIN DESCRIPTION:
South Fork 147.0
END DESCRIPTION:
XS GIS Cut Line= 3
      1450337.50       957986.48      1450251.53       957910.93
      1449767.17       957483.86
#Sta/Elev= 30
  4906.8 1189.61  4924.1 1182.77  4930.7 1180.64  4958.0 1164.78  4967.9 1145.94
  4970.2 1145.94  4973.3 1141.94  5026.7 1141.94  5029.8 1145.94  5041.7 1147.32
  5045.4 1150.93  5048.2 1152.35  5065.2 1150.59  5077.1 1151.06  5098.6 1149.71
  5133.9 1150.61  5154.7 1150.19  5198.1 1151.75  5212.0 1152.90  5219.1 1152.97
  5247.0 1155.81  5259.7 1155.99  5280.0 1157.13  5547.8 1158.80  5568.5 1160.14
  5577.2 1161.27  5590.9 1163.09  5612.3 1168.43  5635.2 1174.70  5667.0 1185.83
#Mann=5,-1,0
  4906.8    0.15       0  4970.2    0.05       0  5029.8    0.15       0
  5154.7    0.08       0  5577.2    0.15       0
#XS Ineff=2,0
       0                 5155.00    0.00 1160.00
Permanent Ineff=
       F       F
Bank Sta=4970.2,5029.8
XS Rating Curve= 0
Exp/Cntr=0.3,0.1

Type RM Length L Ch R = 1,43452,552,552,552
BEGIN DESCRIPTION:
South Fork 145.0
END DESCRIPTION:
XS GIS Cut Line= 4
      1450834.90       957686.99      1450644.76       957574.99
      1450063.31       957246.14      1449881.78       957213.02
#Sta/Elev= 30
  4777.0 1189.95  4791.9 1178.25  4803.3 1167.32  4809.7 1162.75  4821.0 1157.77
  4842.8 1152.98  4870.4 1150.02  4902.0 1147.64  4922.0 1150.91  4934.0 1148.20
  4974.4 1142.90  4977.1 1138.96  5022.9 1138.96  5025.6 1142.90  5035.7 1145.24
  5045.9 1152.10  5053.1 1152.10  5089.5 1152.78  5142.2 1151.07  5248.1 1150.59
  5274.6 1152.06  5373.1 1151.40  5533.4 1154.87  5584.1 1153.88  5645.6 1155.24
  5719.9 1160.17  5767.8 1165.34  5787.9 1169.38  5813.9 1176.48  5850.2 1188.49
#Mann=5,-1,0
  4777.0    0.15       0  4974.4    0.05       0  5025.6    0.15       0
  5053.1    0.08       0  5719.9    0.15       0
#XS Ineff=2,0
    0.00 4922.00 1160.00               0
Permanent Ineff=
       F       F
Bank Sta=4974.4,5025.6
XS Rating Curve= 0
Exp/Cntr=0.3,0.1

Type RM Length L Ch R = 1,42900,681,681,681
BEGIN DESCRIPTION:
South Fork 143.0
END DESCRIPTION:
XS GIS Cut Line= 3
      1450907.76       957082.80      1450813.69       957080.35
      1449879.12       957072.39
#Sta/Elev= 30
  4905.9 1191.93  4911.2 1187.68  4921.0 1181.54  4945.9 1169.27  4956.6 1167.57
  4963.9 1164.12  4971.1 1151.06  4977.6 1141.90  4978.7 1141.81  4981.0 1136.00
  5019.1 1136.00  5021.3 1141.81  5027.2 1141.86  5034.8 1150.88  5072.0 1150.51
  5295.6 1147.25  5397.7 1149.65  5477.5 1150.46  5501.5 1149.61  5515.6 1151.03
  5542.9 1150.72  5758.9 1158.59  5820.9 1163.75  5830.5 1166.06  5843.8 1167.05
  5857.3 1170.04  5868.2 1171.25  5879.4 1174.00  5892.4 1178.67  5934.6 1189.69
#Mann=5,-1,0
  4905.9    0.15       0  4978.7    0.05       0  5021.3    0.15       0
  5072.0    0.08       0  5758.9    0.15       0
#XS Ineff=2,0
       0                 5200.00    0.00 1151.00
Permanent Ineff=
       F       F
Bank Sta=4978.7,5021.3
XS Rating Curve= 0
Exp/Cntr=0.3,0.1

Type RM Length L Ch R = 1,42219,332,332,332
BEGIN DESCRIPTION:
South Fork 141.0
END DESCRIPTION:
XS GIS Cut Line= 3
      1450616.14       956449.96      1450241.11       956890.09
      1449941.67       956910.93
#Sta/Elev= 30
  4912.2 1200.22  4927.6 1194.88  4944.0 1185.47  4945.5 1185.58  4967.2 1149.35
  4971.5 1141.63  4972.3 1140.56  4975.9 1140.52  4978.4 1134.27  5021.6 1134.27
  5024.1 1140.52  5024.9 1140.47  5028.3 1143.38  5032.7 1147.92  5083.6 1144.36
  5106.0 1145.35  5202.3 1145.03  5371.4 1152.60  5473.0 1152.56  5570.5 1154.14
  5609.0 1156.46  5650.8 1162.93  5661.0 1164.52  5672.2 1169.19  5693.8 1174.63
  5711.4 1181.19  5718.6 1182.42  5758.0 1194.05  5779.1 1198.61  5790.6 1201.76
#Mann=5,-1,0
  4912.2    0.15       0  4975.9    0.05       0  5024.1    0.15       0
  5106.0    0.08       0  5650.8    0.15       0
#XS Ineff=2,0
       0                 5066.60    0.00 1148.00
Permanent Ineff=
       F       F
Bank Sta=4975.9,5024.1
XS Rating Curve= 0
Exp/Cntr=0.3,0.1

Type RM Length L Ch R = 1,41887,252,252,252
BEGIN DESCRIPTION:
South Fork 140.0
END DESCRIPTION:
XS GIS Cut Line= 3
      1450316.63       956325.00      1450225.49       956457.80
      1449946.85       956874.45
#Sta/Elev= 30
  4867.5 1190.99  4892.6 1185.01  4915.5 1165.95  4918.9 1161.96  4931.4 1153.14
  4946.3 1145.99  4968.9 1138.22  4983.0 1134.70  4984.8 1130.74  5015.2 1130.74
  5017.0 1134.70  5018.8 1134.78  5022.5 1138.04  5028.2 1134.74  5047.7 1134.75
  5051.5 1142.45  5052.7 1143.06  5085.7 1142.01  5128.0 1142.27  5247.2 1145.76
  5333.3 1146.94  5368.6 1151.20  5384.0 1156.04  5404.2 1162.04  5412.4 1166.32
  5427.8 1170.48  5446.9 1178.93  5462.7 1184.12  5475.5 1186.76  5529.8 1201.45
#Mann=5,-1,0
  4867.5    0.15       0  4983.0    0.05       0  5017.0    0.15       0
  5128.0    0.08       0  5384.0    0.15       0
#XS Ineff=2,0
       0                 5100.00    0.00 1146.00
Permanent Ineff=
       F       F
Bank Sta=4983,5017
XS Rating Curve= 0
Exp/Cntr=0.3,0.1

Type RM Length L Ch R = 1,41635,235,235,235
BEGIN DESCRIPTION:
South Fork 139.0
END DESCRIPTION:
XS GIS Cut Line= 3
      1450152.58       956244.26      1450006.74       956345.82
      1449600.52       956650.49
#Sta/Elev= 30
  4831.9 1169.83  4845.9 1159.29  4857.1 1153.83  4873.5 1147.71  4889.0 1137.44
  4905.6 1136.61  4935.4 1139.64  4971.2 1139.68  4987.2 1133.50  4988.6 1129.58
  5011.4 1129.58  5012.8 1133.50  5032.8 1133.81  5035.7 1136.62  5037.1 1145.15
  5063.4 1144.56  5082.8 1142.61  5121.9 1140.31  5145.8 1133.84  5169.9 1133.96
  5182.0 1140.23  5202.0 1140.68  5262.6 1144.16  5376.5 1142.26  5405.7 1143.22
  5430.6 1145.05  5454.4 1148.56  5480.0 1153.76  5512.0 1167.67  5517.4 1170.74
#Mann=5,-1,0
  4831.9    0.15       0  4987.2    0.05       0  5012.8    0.15       0
  5202.0    0.08       0  5454.4    0.15       0
#XS Ineff=2,0
    0.00 4900.00 1148.00 5262.00    0.00 1148.00
Permanent Ineff=
       F       F
Bank Sta=4987.2,5012.8
XS Rating Curve= 0
Exp/Cntr=0.3,0.1

Type RM Length L Ch R = 1,41400,220,220,220
BEGIN DESCRIPTION:
South Fork 138.0
END DESCRIPTION:
XS GIS Cut Line= 3
      1450025.00       956075.00      1449908.42       956132.76
      1449402.55       956436.98
#Sta/Elev= 30
  4869.9 1176.56  4897.4 1164.80  4939.4 1135.33  4954.1 1134.74  4967.0 1135.44
  4974.1 1134.35  4985.8 1131.28  4987.3 1128.28  5012.7 1128.28  5014.2 1131.28
  5026.6 1132.54  5034.4 1140.69  5077.8 1139.90  5106.7 1141.19  5116.6 1140.53
  5145.3 1132.29  5169.8 1132.29  5171.8 1137.23  5176.7 1139.32  5228.7 1141.57
  5411.6 1142.53  5428.8 1141.73  5482.5 1141.54  5500.1 1143.76  5519.6 1151.66
  5522.5 1152.44  5525.7 1151.58  5571.7 1171.87  5583.1 1173.65  5590.3 1173.99
#Mann=5,-1,0
  4869.9    0.15       0  4985.8    0.05       0  5014.2    0.15       0
  5228.7    0.08       0  5411.6    0.15       0
#XS Ineff=2,0
       0                 5300.00    0.00 1146.00
Permanent Ineff=
       F       F
Bank Sta=4985.8,5014.2
XS Rating Curve= 0
Exp/Cntr=0.3,0.1

Type RM Length L Ch R = 1,41180,253,253,253
BEGIN DESCRIPTION:
South Fork 137.0
END DESCRIPTION:
XS GIS Cut Line= 3
      1450071.86       955923.95      1449918.20       955921.34
      1449506.73       955960.41
#Sta/Elev= 30
  4837.0 1171.71  4852.7 1170.60  4866.9 1168.26  4906.8 1165.33  4954.9 1142.55
  4976.7 1133.09  4985.8 1130.71  4987.3 1127.71  5012.7 1127.71  5014.2 1130.71
  5018.8 1131.72  5021.2 1139.44  5021.7 1140.01  5030.9 1142.09  5045.3 1142.33
  5064.6 1141.83  5071.1 1142.23  5102.1 1141.88  5141.2 1142.97  5158.6 1142.88
  5173.7 1143.80  5207.3 1144.83  5224.0 1144.60  5249.2 1146.03  5260.7 1146.25
  5318.7 1144.65  5329.7 1147.46  5349.0 1154.06  5378.0 1159.59  5404.0 1167.28
#Mann=3,-1,0
  4837.0    0.15       0  4985.8    0.05       0  5014.2    0.15       0
Bank Sta=4985.8,5014.2
XS Rating Curve= 0
Exp/Cntr=0.3,0.1

Type RM Length L Ch R = 1,40927,557,557,557
BEGIN DESCRIPTION:
South Fork 136.0
END DESCRIPTION:
XS GIS Cut Line= 3
      1450144.74       955788.52      1449957.26       955684.37
      1449819.24       955608.85
#Sta/Elev= 30
  4775.3 1160.95  4789.1 1160.59  4807.2 1159.63  4847.7 1152.09  4852.7 1150.47
  4858.9 1149.01  4863.0 1147.63  4892.2 1140.48  4927.1 1138.46  4943.7 1139.62
  4954.0 1138.27  4960.5 1134.49  4974.4 1131.73  4985.8 1130.60  4987.3 1126.55
  5012.7 1126.55  5014.2 1130.60  5027.5 1131.05  5032.4 1133.84  5045.8 1143.93
  5055.8 1144.79  5066.5 1146.41  5076.1 1148.38  5082.5 1149.08  5115.2 1155.61
  5117.2 1156.17  5126.5 1161.23  5130.1 1162.73  5139.1 1165.76  5147.1 1169.00
#Mann=3,-1,0
  4775.3    0.15       0  4985.8    0.05       0  5014.2    0.15       0
Bank Sta=4985.8,5014.2
XS Rating Curve= 0
Exp/Cntr=0.3,0.1

Type RM Length L Ch R = 1,40370,410,410,410
BEGIN DESCRIPTION:
South Fork 135.0
END DESCRIPTION:
XS GIS Cut Line= 3
      1450186.42       955785.96      1450246.32       955270.30
      1450256.74       955150.48
#Sta/Elev= 30
  4448.7 1157.56  4493.2 1154.58  4520.2 1153.97  4532.2 1152.72  4548.2 1152.52
  4565.7 1151.40  4635.4 1148.61  4717.1 1146.15  4728.7 1145.46  4761.2 1143.93
  4780.3 1142.64  4806.6 1141.15  4821.1 1140.54  4835.4 1140.11  4870.5 1139.65
  4891.6 1139.69  4927.3 1139.44  4953.6 1140.49  4958.8 1137.65  4976.0 1129.62
  4984.4 1128.56  4986.0 1125.56  5014.0 1125.56  5015.6 1128.56  5026.1 1139.89
  5043.9 1157.25  5058.2 1168.76  5070.0 1180.36  5087.1 1193.84  5088.1 1194.33
#Mann=4,-1,0
  4448.7    0.08       0  4891.6    0.15       0  4984.4    0.05       0
  5015.6    0.15       0
Bank Sta=4984.4,5015.6
XS Rating Curve= 0
Exp/Cntr=0.3,0.1

Type RM Length L Ch R = 1,39960,360,360,360
BEGIN DESCRIPTION:
South Fork 133.0
END DESCRIPTION:
XS GIS Cut Line= 3
      1450574.45       956022.86      1450649.97       955291.14
      1450665.59       955147.90
#Sta/Elev= 30
  4265.8 1153.49  4277.3 1151.75  4335.1 1147.74  4392.5 1145.60  4517.7 1142.17
  4572.0 1141.16  4696.4 1140.54  4758.6 1141.25  4800.9 1140.95  4858.1 1138.25
  4888.5 1136.84  4890.4 1136.21  4927.4 1136.10  4935.9 1137.00  4948.2 1136.98
  4963.8 1138.32  4965.3 1137.29  4977.1 1133.09  4981.8 1129.69  4984.1 1128.63
  4985.7 1124.58  5014.3 1124.58  5019.9 1128.63  5028.4 1132.80  5045.9 1138.52
  5054.4 1141.91  5073.8 1147.75  5101.1 1152.59  5124.3 1154.85  5145.5 1155.81
#Mann=4,-1,0
  4265.8    0.08       0  4858.1    0.15       0  4984.1    0.05       0
  5019.9    0.15       0
Bank Sta=4984.1,5019.9
XS Rating Curve= 0
Exp/Cntr=0.3,0.1

Type RM Length L Ch R = 1,39600,275,275,275
BEGIN DESCRIPTION:
South Fork 132.0
END DESCRIPTION:
XS GIS Cut Line= 4
      1451202.05       955671.34      1450988.74       955342.11
      1450845.28       955147.91      1450655.18       955054.16
#Sta/Elev= 30
  4607.7 1191.18  4637.8 1183.46  4666.7 1174.68  4685.7 1167.33  4720.4 1150.03
  4746.3 1138.50  4756.7 1136.55  4797.6 1134.97  4847.5 1135.67  4944.6 1137.34
  4957.4 1132.90  4967.7 1131.46  4975.8 1127.32  4985.5 1126.19  4987.0 1123.19
  5013.0 1123.19  5014.5 1126.19  5032.8 1127.19  5033.4 1130.16  5038.2 1131.48
  5089.0 1131.30  5110.1 1132.09  5142.8 1135.64  5187.3 1136.48  5233.5 1138.77
  5255.0 1140.88  5304.8 1142.96  5337.2 1146.91  5349.3 1147.30  5453.4 1160.46
#Mann=5,-1,0
  4607.7    0.14       0  4847.5    0.08       0  4985.5    0.05       0
  5014.5    0.08       0  5089.0    0.15       0
#XS Ineff=2,0
    0.00 4900.00 1137.50 5110.00    0.00 1139.00
Permanent Ineff=
       F       F
Bank Sta=4985.5,5014.5
XS Rating Curve= 0
Exp/Cntr=0.3,0.1

Type RM Length L Ch R = 1,39325,549,549,549
BEGIN DESCRIPTION:
South Fork 131.0
END DESCRIPTION:
XS GIS Cut Line= 3
      1451415.61       955202.61      1451332.26       955132.28
      1450626.54       955022.91
#Sta/Elev= 30
  4586.1 1160.38  4605.3 1157.15  4630.8 1155.61  4647.8 1150.46  4665.3 1146.28
  4710.5 1131.46  4722.4 1132.82  4765.2 1135.15  4803.1 1134.21  4815.5 1134.14
  4849.5 1134.64  4873.9 1135.93  4883.8 1135.52  4897.0 1131.23  4907.2 1130.18
  4919.3 1127.59  4923.5 1126.05  4946.8 1125.95  4981.2 1125.80  4983.1 1122.05
  5016.9 1122.05  5018.9 1126.20  5041.1 1126.28  5042.9 1127.27  5049.8 1136.20
  5050.3 1137.43  5173.3 1138.92  5231.7 1142.83  5345.9 1157.15  5409.3 1167.09
#Mann=6,-1,0
  4586.1    0.14       0  4803.1    0.15       0  4815.5    0.08       0
  4946.8    0.15       0  4981.2    0.05       0  5018.9    0.15       0
#XS Ineff=2,0
    0.00 4765.00 1136.50               0
Permanent Ineff=
       F       F
Bank Sta=4981.2,5018.9
XS Rating Curve= 0
Exp/Cntr=0.3,0.1

Type RM Length L Ch R = 1,38776,433,433,433
BEGIN DESCRIPTION:
South Fork 130.0
END DESCRIPTION:
XS GIS Cut Line= 3
      1451730.69       954819.79      1451673.40       954877.07
      1450647.36       954913.53
#Sta/Elev= 30
  4720.9 1176.06  4759.3 1168.65  4768.9 1167.72  4817.9 1155.76  4822.3 1155.75
  4880.2 1143.69  4909.6 1136.37  4924.0 1134.76  4946.3 1135.01  4971.3 1126.01
  4981.4 1123.95  4984.1 1123.90  4985.7 1120.01  5014.3 1120.01  5016.0 1123.90
  5026.7 1124.07  5030.2 1128.93  5036.2 1133.14  5055.6 1132.45  5103.7 1134.92
  5251.3 1136.56  5347.5 1135.47  5358.5 1134.36  5388.3 1134.08  5396.9 1134.85
  5511.2 1136.02  5609.3 1140.68  5672.4 1144.68  5769.5 1156.13  5828.6 1166.27
#Mann=4,-1,0
  4720.9    0.14       0  4981.4    0.15       0  4984.1    0.05       0
  5016.0    0.15       0
#XS Ineff=2,0
       0                 5067.80    0.00 1133.00
Permanent Ineff=
       F       F
Bank Sta=4984.1,5016
XS Rating Curve= 0
Exp/Cntr=0.3,0.1

Type RM Length L Ch R = 1,38343,543,543,543
BEGIN DESCRIPTION:
South Fork 127.0
END DESCRIPTION:
XS GIS Cut Line= 3
      1451355.70       954457.80      1450939.03       954814.57
      1450636.95       954824.99
#Sta/Elev= 30
  4843.7 1156.99  4854.4 1156.01  4869.0 1151.73  4883.3 1145.96  4915.9 1135.97
  4934.8 1134.06  4953.5 1126.28  4964.8 1126.63  4967.4 1123.18  4973.9 1122.77
  4976.6 1118.77  5023.4 1118.77  5026.1 1122.77  5030.6 1126.28  5042.2 1131.14
  5043.2 1132.17  5047.2 1132.34  5071.3 1132.85  5088.8 1132.16  5182.5 1131.69
  5216.3 1133.26  5280.7 1132.97  5354.0 1135.49  5377.9 1135.43  5505.5 1141.41
  5541.3 1145.53  5564.2 1146.27  5612.5 1152.97  5661.5 1162.49  5694.5 1172.86
#Mann=4,-1,0
  4843.7    0.14       0  4883.3    0.15       0  4973.9    0.05       0
  5026.1    0.15       0
Bank Sta=4973.9,5026.1
XS Rating Curve= 0
Exp/Cntr=0.3,0.1

Type RM Length L Ch R = 1,37800,381,381,381
BEGIN DESCRIPTION:
South Fork 126.0
END DESCRIPTION:
XS GIS Cut Line= 3
      1451428.63       954280.72      1450817.02       954302.46
      1450467.72       954304.16
#Sta/Elev= 30
  4388.0 1161.00  4407.1 1158.12  4451.6 1155.18  4501.1 1150.12  4523.0 1146.20
  4610.5 1136.58  4679.8 1131.13  4851.8 1130.89  4877.1 1131.42  4916.3 1128.18
  4927.0 1129.43  4962.7 1129.44  4974.3 1121.68  4985.5 1120.56  4987.0 1117.56
  5013.0 1117.56  5014.5 1120.56  5029.9 1121.56  5060.4 1129.04  5174.6 1127.25
  5223.7 1128.67  5252.3 1127.78  5278.7 1128.77  5298.4 1131.59  5312.2 1140.45
  5321.2 1148.47  5334.1 1162.78  5339.6 1165.89  5344.3 1172.02  5349.3 1176.78
#Mann=5,-1,0
  4388.0    0.15       0  4610.5    0.08       0  4851.8    0.15       0
  4985.5    0.05       0  5014.5    0.15       0
#XS Ineff=2,0
       0                 5200.00    0.00 1130.00
Permanent Ineff=
       F       F
Bank Sta=4985.5,5014.5
XS Rating Curve= 0
Exp/Cntr=0.3,0.1

Type RM Length L Ch R = 1,37419,1148,1148,1148
BEGIN DESCRIPTION:
South Fork 125.0
END DESCRIPTION:
XS GIS Cut Line= 4
      1451345.32       953908.31      1451217.68       953957.80
      1450415.59       953976.03      1450350.49       954056.76
#Sta/Elev= 30
  4288.7 1165.38  4311.6 1162.46  4359.0 1152.40  4388.1 1143.63  4415.8 1133.02
  4452.3 1125.12  4525.7 1126.97  4573.8 1127.76  4704.5 1127.19  4750.3 1127.06
  4777.6 1124.41  4791.9 1124.66  4829.2 1127.23  4961.7 1128.79  4967.3 1120.66
  4976.8 1120.37  4979.2 1116.37  5020.8 1116.37  5023.2 1120.37  5023.4 1120.37
  5023.8 1125.28  5027.9 1127.87  5036.7 1126.73  5078.3 1126.40  5103.5 1128.53
  5125.4 1133.07  5164.7 1146.62  5227.9 1152.49  5271.4 1162.06  5331.6 1171.95
#Mann=5,-1,0
  4288.7    0.15       0  4525.7    0.08       0  4704.5    0.15       0
  4976.8    0.05       0  5023.2    0.15       0
#XS Ineff=2,0
    0.00 4750.00 1131.00               0
Permanent Ineff=
       F       F
Bank Sta=4976.8,5023.2
XS Rating Curve= 0
Exp/Cntr=0.3,0.1

Type RM Length L Ch R = 1,36271,606,606,606
BEGIN DESCRIPTION:
South Fork 121.0
END DESCRIPTION:
XS GIS Cut Line= 3
      1451337.49       953783.34      1451149.97       953671.34
      1450655.19       953314.59
#Sta/Elev= 30
  4769.0 1161.74  4821.6 1157.25  4850.0 1153.82  4861.9 1151.72  4890.9 1144.77
  4907.4 1137.43  4926.5 1126.75  4933.7 1125.25  4944.2 1125.67  4948.6 1125.15
  4959.0 1121.64  4968.7 1120.36  4978.1 1116.74  4980.4 1112.74  5019.7 1112.74
  5021.9 1116.74  5022.9 1116.81  5023.2 1118.44  5033.9 1126.07  5061.1 1124.58
  5149.5 1126.65  5215.1 1129.85  5351.6 1134.06  5391.3 1136.44  5398.0 1136.28
  5409.0 1137.39  5477.6 1139.34  5519.0 1141.97  5567.8 1143.79  5597.4 1146.10
#Mann=4,-1,0
  4769.0    0.15       0  4978.1    0.05       0  5021.9    0.15       0
  5061.1    0.08       0
Bank Sta=4978.1,5021.9
XS Rating Curve= 0
Exp/Cntr=0.3,0.1

Type RM Length L Ch R = 1,35665,364,364,364
BEGIN DESCRIPTION:
South Fork 119.0
END DESCRIPTION:
XS GIS Cut Line= 4
      1451915.61       953426.56      1451470.28       953166.14
      1450995.99       952916.51      1450920.77       952835.37
#Sta/Elev= 30
  4472.6 1163.82  4537.2 1158.11  4580.2 1152.68  4620.0 1146.33  4629.9 1143.40
  4652.1 1140.66  4668.7 1135.55  4731.3 1128.24  4833.0 1123.43  4930.1 1123.29
  4959.0 1124.54  4966.2 1115.04  4970.8 1114.98  4973.8 1110.98  5026.2 1110.98
  5029.2 1114.98  5038.6 1121.58  5041.5 1123.91  5069.0 1120.96  5397.3 1127.05
  5428.7 1127.96  5465.5 1132.81  5502.4 1133.14  5505.5 1135.30  5509.3 1135.87
  5520.8 1135.19  5538.0 1137.47  5571.8 1144.50  5591.3 1150.68  5635.1 1160.59
#Mann=7,-1,0
  4472.6    0.15       0  4731.3    0.08       0  4930.1    0.15       0
  4970.8    0.05       0  5029.2    0.15       0  5038.6    0.08       0
  5397.3    0.08       0
Bank Sta=4970.8,5029.2
XS Rating Curve= 0
Exp/Cntr=0.3,0.1

Type RM Length L Ch R = 1,35301,363,363,363
BEGIN DESCRIPTION:
South Fork 118.0
END DESCRIPTION:
XS GIS Cut Line= 3
      1452074.47       953215.63      1451590.07       952861.45
      1451379.16       952692.20
#Sta/Elev= 30
  4334.6 1152.94  4384.8 1145.57  4426.3 1140.83  4452.5 1134.54  4474.7 1131.37
  4490.9 1127.79  4518.9 1124.84  4539.2 1123.80  4590.6 1123.17  4619.7 1121.90
  4729.0 1123.14  4792.6 1121.59  4849.2 1122.59  4899.4 1121.60  4937.8 1122.90
  4948.1 1119.05  4968.5 1113.98  4972.3 1113.97  4975.1 1109.97  5024.9 1109.97
  5027.7 1113.97  5028.3 1113.98  5031.9 1120.42  5035.7 1122.61  5093.6 1121.64
  5114.3 1134.29  5132.0 1147.29  5163.0 1162.30  5192.3 1178.46  5205.1 1182.52
#Mann=5,-1,0
  4334.6    0.15       0  4590.6    0.08       0  4899.4    0.15       0
  4972.3    0.05       0  5027.7    0.15       0
#XS Ineff=2,0
    0.00 4849.00 1124.00               0
Permanent Ineff=
       F       F
Bank Sta=4972.3,5027.7
XS Rating Curve= 0
Exp/Cntr=0.3,0.1

Type RM Length L Ch R = 1,34938,456,456,456
BEGIN DESCRIPTION:
South Fork 117.0
END DESCRIPTION:
XS GIS Cut Line= 3
      1452347.88       953072.38      1452269.76       953022.91
      1451524.97       952474.98
#Sta/Elev= 30
  4335.8 1166.15  4407.8 1148.54  4446.2 1141.68  4483.8 1136.68  4504.8 1131.62
  4531.1 1128.63  4583.9 1124.74  4614.2 1121.92  4651.1 1122.48  4701.6 1120.11
  4786.4 1121.70  4863.2 1120.61  4953.0 1121.49  4956.7 1119.86  4972.3 1113.75
  4975.1 1107.84  5024.9 1107.84  5027.7 1113.75  5029.5 1113.84  5030.2 1119.67
  5030.7 1122.63  5119.3 1121.60  5139.9 1122.47  5213.4 1120.65  5262.7 1124.51
  5279.6 1127.18  5298.0 1133.21  5317.8 1146.15  5338.6 1156.63  5352.9 1161.27
#Mann=5,-1,0
  4335.8    0.15       0  4583.9    0.08       0  4956.7    0.15       0
  4972.3    0.05       0  5027.7    0.15       0
#XS Ineff=2,0
    0.00 4763.00 1125.00 5150.00    0.00 1125.00
Permanent Ineff=
       F       F
Bank Sta=4972.3,5027.7
XS Rating Curve= 0
Exp/Cntr=0.3,0.1

Type RM Length L Ch R = 1,34482,409,409,409
BEGIN DESCRIPTION:
South Fork 115.0
END DESCRIPTION:
XS GIS Cut Line= 3
      1452358.31       953002.08      1452209.86       952879.68
      1452032.78       952259.88
#Sta/Elev= 30
  4282.8 1159.16  4331.4 1144.96  4361.4 1137.34  4430.5 1123.13  4465.0 1123.92
  4496.4 1121.79  4522.2 1120.94  4550.9 1121.34  4585.2 1120.46  4666.6 1121.70
  4762.9 1120.75  4812.0 1121.79  4838.9 1118.18  4855.9 1117.82  4913.5 1119.65
  4936.1 1117.25  4956.9 1118.40  4958.8 1117.90  4965.1 1113.68  4978.1 1113.50
  4980.4 1107.68  5019.7 1107.68  5021.9 1113.50  5038.9 1120.51  5044.5 1123.41
  5048.7 1123.82  5068.7 1130.77  5084.2 1140.15  5112.5 1152.34  5119.8 1156.43
#Mann=5,-1,0
  4282.8    0.15       0  4585.2    0.08       0  4762.9    0.15       0
  4978.1    0.05       0  5021.9    0.15       0
#XS Ineff=2,0
    0.00 4750.00 1122.00               0
Permanent Ineff=
       F       F
Bank Sta=4978.1,5021.9
XS Rating Curve= 0
Exp/Cntr=0.3,0.1
