HEC-RAS study Grassy Creek.prj: Grassy Creek Limited Detail Study

--- Grassy Creek.g01 (geometry) --- (continued)

Type RM Length L Ch R = 1,40640,402,402,402
BEGIN DESCRIPTION:
Grassy Creek 73.0
END DESCRIPTION:
XS GIS Cut Line= 3
      1571748.56       942457.52      1571242.84       942306.88
      1571167.52       942255.78
#Sta/Elev= 30
  4662.3  972.89  4697.9  967.09  4721.1  965.07  4728.4  963.25  4752.6  959.36
  4782.5  955.48  4795.8  952.94  4833.2  948.23  4864.9  941.80  4888.2  936.36
  4898.1  936.62  4936.8  935.59  4959.6  935.91  4983.0  935.44  4993.5  934.45
  4996.8  929.45  5003.3  929.45  5006.5  934.45  5031.5  935.54  5059.5  938.41
  5073.7  938.88  5079.2  939.77  5098.2  945.02  5124.7  949.21  5159.7  955.94
  5198.2  965.46  5216.2  968.74  5224.3  971.58  5233.9  973.91  5281.0  984.19
#Mann=4,-1,0
  4662.3    0.15       0  4864.9    0.13       0  4993.5    0.05       0
  5006.5    0.13       0
Bank Sta=4993.5,5006.5
XS Rating Curve= 0
Exp/Cntr=0.3,0.1

Type RM Length L Ch R = 1,40238,284,284,284
BEGIN DESCRIPTION:
Grassy Creek 72.0
END DESCRIPTION:
XS GIS Cut Line= 3
      1571869.64       942247.68      1571794.32       942067.45
      1571315.50       941916.81
#Sta/Elev= 30
  4505.8  977.49  4531.1  975.54  4588.5  965.45  4611.3  960.06  4657.1  947.14
  4679.9  941.93  4711.9  937.94  4726.6  936.86  4821.6  935.41  4831.6  934.52
  4850.2  934.66  4876.4  936.59  4900.1  934.09  4931.0  934.12  4959.3  935.96
  4969.4  934.02  4993.0  931.80  4996.5  926.80  5003.5  926.80  5007.0  931.80
  5011.3  931.91  5029.9  936.07  5062.0  936.90  5078.3  942.49  5087.1  947.64
  5101.9  954.00  5126.3  962.50  5157.4  968.52  5181.3  976.28  5203.1  981.54
#Mann=3,-1,0
  4505.8    0.13       0  4993.0    0.05       0  5007.0    0.13       0
#XS Ineff=2,0
    0.00 4880.30  944.60               0
Permanent Ineff=
       F       F
Bank Sta=4993,5007
XS Rating Curve= 0
Exp/Cntr=0.5,0.3

Type RM Length L Ch R = 1,39954,88,88,88
BEGIN DESCRIPTION:
Pinnacle Hotel Rd (GC) us
END DESCRIPTION:
XS GIS Cut Line= 5
      1572159.63       941716.15      1571866.11       941751.87
      1571682.88       941734.79      1571463.93       941683.55
      1571344.35       941641.61
#Sta/Elev= 30
  4435.3  958.68  4445.9  959.29  4464.1  957.41  4493.4  959.67  4508.5  956.12
  4528.8  956.46  4564.8  953.36  4593.7  952.52  4603.1  950.33  4609.9  951.77
  4621.3  949.46  4665.9  949.32  4709.4  944.86  4729.8  944.94  4738.0  943.19
  4814.8  937.09  4846.8  935.65  4868.4  935.89  4873.7  933.94  4915.0  929.94
  4982.5  930.05  4983.0  924.95  5017.0  924.95  5017.5  930.05  5049.2  936.66
  5083.9  938.38  5135.5  944.26  5236.3  961.43  5248.6  962.37  5266.6  961.12
#Mann=5,-1,0
  4435.3    0.13       0  4738.0    0.07       0  4873.7    0.13       0
  4982.5    0.05       0  5017.5    0.13       0
#XS Ineff=2,0
    0.00 4971.50  937.20 5028.50    0.00  937.80
Permanent Ineff=
       F       F
Bank Sta=4982.5,5017.5
XS Rating Curve= 0
Exp/Cntr=0.5,0.3

Type RM Length L Ch R =2,39913,,,
BEGIN DESCRIPTION:
Pinnacle Hotel Rd (GC) TOR
Structure ID: LDS_GC_06
Approximate Survey Structure
END DESCRIPTION:
Bridge Culvert--1,0,-1,-1,0
Deck Dist Width WeirC Skew NumUp NumDn MinLoCord MaxHiCord MaxSubmerge Is_Ogee
16,50,3,,14,14,,,0.95,0,1,1,,,
  4336.0  4435.8  4521.1  4609.3  4704.5  4775.2  4830.0  4881.6  4950.0  5017.0
  5057.4  5158.7  5249.4  5298.2
  955.19  950.57  946.30  942.61  939.42  937.23  936.65  936.64  937.20  937.20
  939.00  945.08  955.24  961.03
  905.00  905.00  905.00  905.00  905.00  905.00  905.00  905.00  905.00  905.00
  905.00  905.00  905.00  905.00
  4336.0  4435.8  4521.1  4609.3  4704.5  4775.2  4830.0  4881.6  4950.0  5017.0
  5057.4  5158.7  5249.4  5298.2
  955.19  950.57  946.30  942.61  939.42  937.23  936.65  936.64  937.20  937.20
  939.00  945.08  955.24  961.03
  904.75  904.75  904.75  904.75  904.75  904.75  904.75  904.75  904.75  904.75
  904.75  904.75  904.75  904.75
Culvert=2,8,12,50,0.012,0.4,1,8,1,925,4993.5,924.75,4993.5,Culvert #1,0,16
Culvert Bottom n=0.012
Culvert Bottom Depth=0
Culvert Depth Blocked=0
Culvert=2,8,12,50,0.012,0.4,1,8,1,925,5006.5,924.75,5006.5,Culvert #2,0,16
Culvert Bottom n=0.012
Culvert Bottom Depth=0
Culvert Depth Blocked=0
BC Design=,,0,,0,,,,,,

Type RM Length L Ch R = 1,39866,301,301,301
BEGIN DESCRIPTION:
Pinnacle Hotel Rd (GC) ds
END DESCRIPTION:
XS GIS Cut Line= 5
      1572235.72       941633.85      1571884.74       941678.89
      1571713.93       941657.15      1571527.60       941613.67
      1571330.37       941565.53
#Sta/Elev= 30
  4365.4  954.85  4389.8  951.99  4429.0  953.29  4469.9  950.05  4481.8  951.90
  4492.1  949.37  4499.7  950.82  4511.0  947.78  4556.4  948.84  4581.2  945.95
  4592.7  946.99  4675.3  941.37  4732.3  940.51  4743.8  941.02  4827.5  934.00
  4867.2  933.23  4891.4  934.40  4916.3  932.57  4944.0  934.70  4954.2  931.96
  4982.5  929.85  4983.0  924.75  5017.0  924.75  5017.5  929.85  5024.7  935.29
  5032.6  936.21  5177.5  948.17  5212.4  952.64  5226.2  952.69  5285.8  960.66
#Mann=4,-1,0
  4365.4    0.13       0  4732.3    0.07       0  4982.5    0.05       0
  5017.5    0.13       0
#XS Ineff=2,0
    0.00 4965.50  937.20 5034.50    0.00  937.76
Permanent Ineff=
       F       F
Bank Sta=4982.5,5017.5
XS Rating Curve= 0
Exp/Cntr=0.5,0.3

Type RM Length L Ch R = 1,39565,214,214,214
BEGIN DESCRIPTION:
Grassy Creek 71.0
END DESCRIPTION:
XS GIS Cut Line= 4
      1572286.62       941602.05      1572060.65       941564.39
      1571708.24       941357.25      1571640.97       941260.39
#Sta/Elev= 30
  4404.1  958.89  4438.5  957.84  4464.0  956.03  4472.3  954.10  4488.5  954.01
  4504.0  949.90  4514.0  950.23  4522.9  953.30  4568.4  950.86  4582.5  949.06
  4593.6  949.48  4649.2  947.40  4701.6  941.54  4730.8  936.95  4769.4  932.79
  4820.6  932.46  4928.2  929.58  4962.3  930.16  4993.0  928.00  4996.5  923.00
  5003.5  923.00  5007.0  928.00  5022.4  928.00  5044.9  932.57  5051.6  936.68
  5065.8  940.63  5073.0  944.23  5087.1  948.90  5129.5  959.32  5159.9  964.11
#Mann=5,-1,0
  4404.1    0.13       0  4730.8    0.07       0  4928.2    0.13       0
  4993.0    0.05       0  5007.0    0.13       0
Bank Sta=4993,5007
XS Rating Curve= 0
Exp/Cntr=0.3,0.1

Type RM Length L Ch R = 1,39351,690,690,690
BEGIN DESCRIPTION:
Grassy Creek 70.0
END DESCRIPTION:
XS GIS Cut Line= 3
      1572267.70       941350.36      1572093.65       941309.75
      1571734.01       941164.73
#Sta/Elev= 30
  4600.6  960.70  4616.6  958.52  4656.2  955.10  4688.8  950.57  4718.7  945.67
  4744.4  942.49  4762.7  938.32  4779.3  933.56  4786.7  931.85  4789.6  931.64
  4817.0  929.98  4847.5  929.45  4854.2  928.50  4898.6  928.09  4906.7  927.47
  4939.8  924.68  4954.3  924.74  4962.0  925.76  4976.5  929.28  4993.0  927.48
  4996.5  922.48  5003.5  922.48  5007.0  927.48  5034.4  931.23  5044.4  934.22
  5057.6  941.73  5066.7  946.34  5098.2  958.24  5119.5  963.14  5167.1  972.18
#Mann=5,-1,0
  4600.6    0.13       0  4789.6    0.07       0  4906.7    0.13       0
  4993.0    0.05       0  5007.0    0.13       0
Bank Sta=4993,5007
XS Rating Curve= 0
Exp/Cntr=0.3,0.1

Type RM Length L Ch R = 1,38661,655,655,655
BEGIN DESCRIPTION:
Grassy Creek 69.0
END DESCRIPTION:
XS GIS Cut Line= 4
      1572644.67       940613.68      1572424.29       940712.28
      1572348.88       940729.68      1571989.22       940712.28
#Sta/Elev= 30
  4541.3  961.41  4564.9  958.12  4579.5  956.96  4605.4  953.43  4642.3  949.37
  4681.9  942.71  4749.1  934.46  4780.4  931.53  4809.6  929.92  4884.9  926.88
  4904.3  926.51  4934.4  924.76  4950.9  925.50  4962.5  924.76  4976.0  922.67
  4993.0  922.03  4996.5  917.03  5003.5  917.03  5007.0  922.03  5024.8  924.81
  5026.2  925.50  5051.3  930.84  5086.0  939.04  5102.7  943.45  5116.4  946.41
  5130.8  948.91  5157.9  952.59  5184.0  956.99  5199.0  960.15  5220.2  963.93
#Mann=5,-1,0
  4541.3    0.13       0  4749.1    0.07       0  4809.6    0.13       0
  4993.0    0.05       0  5007.0    0.13       0
Bank Sta=4993,5007
XS Rating Curve= 0
Exp/Cntr=0.3,0.1

Type RM Length L Ch R = 1,38006,252,252,252
BEGIN DESCRIPTION:
Grassy Creek 68.0
END DESCRIPTION:
XS GIS Cut Line= 3
      1572656.35       940080.01      1572493.90       940039.39
      1571693.36       940167.02
#Sta/Elev= 30
  4524.6  953.86  4549.4  952.54  4565.3  950.15  4587.2  948.51  4592.4  948.88
  4610.8  946.85  4647.7  939.64  4662.0  938.64  4681.8  934.14  4716.4  930.13
  4742.8  927.19  4798.9  924.78  4953.1  921.29  4993.0  918.43  4996.5  913.43
  5003.5  913.43  5007.0  918.43  5036.5  921.64  5075.4  922.98  5085.4  922.54
  5106.8  922.47  5116.9  923.68  5136.1  923.17  5155.0  925.55  5170.2  925.70
  5227.4  930.92  5271.4  937.24  5335.7  946.39  5442.4  960.27  5502.7  966.41
#Mann=8,-1,0
  4524.6    0.13       0  4716.4    0.07       0  4953.1    0.13       0
  4993.0    0.05       0  5007.0    0.13       0  5085.4    0.07       0
  5271.4    0.13       0  5335.7    0.07       0
Bank Sta=4993,5007
XS Rating Curve= 0
Exp/Cntr=0.3,0.1

Type RM Length L Ch R = 1,37754,237,237,237
BEGIN DESCRIPTION:
Grassy Creek 67.5
END DESCRIPTION:
XS GIS Cut Line= 3
      1572353.04       939673.93      1572040.06       939901.40
      1571774.98       940074.13
#Sta/Elev= 30
  4657.5  959.63  4663.2  957.04  4680.2  946.96  4695.2  939.84  4698.5  936.99
  4703.3  934.01  4724.7  924.04  4753.4  922.63  4760.5  922.06  4786.8  921.73
  4802.5  922.29  4846.2  920.84  4879.0  920.95  4935.4  919.89  4958.9  920.97
  4976.3  918.91  4993.0  916.93  4996.5  911.93  5003.5  911.93  5007.0  916.93
  5044.7  921.32  5069.9  919.29  5085.1  919.47  5129.9  920.19  5165.4  929.35
  5175.5  930.84  5197.3  932.97  5260.5  941.29  5314.1  949.28  5360.8  954.00
#Mann=6,-1,0
  4657.5    0.13       0  4753.4    0.07       0  4976.3    0.13       0
  4993.0    0.05       0  5007.0    0.13       0  5085.1    0.07       0
#XS Ineff=2,0
    0.00 4841.80  928.66               0
Permanent Ineff=
       F       F
Bank Sta=4993,5007
XS Rating Curve= 0
Exp/Cntr=0.3,0.1

Type RM Length L Ch R = 1,37517,685,685,685
BEGIN DESCRIPTION:
Grassy Creek 67.0
END DESCRIPTION:
XS GIS Cut Line= 4
      1572192.72       939525.60      1571912.16       939724.33
      1571730.94       939920.16      1571649.08       940034.19
#Sta/Elev= 30
  4614.4  973.09  4663.3  953.75  4685.6  945.83  4716.1  931.54  4727.5  927.83
  4746.4  920.55  4748.3  919.93  4764.5  919.08  4811.8  918.89  4851.1  919.60
  4894.6  918.27  4945.2  919.26  4963.3  920.21  4993.0  915.05  4996.5  910.05
  5003.5  910.05  5007.0  915.05  5032.9  918.80  5044.9  918.60  5057.9  919.69
  5106.6  932.37  5151.5  933.64  5174.1  935.18  5222.2  939.83  5266.2  945.94
  5306.0  952.76  5316.3  957.64  5341.1  957.85  5352.8  959.39  5365.4  959.59
#Mann=7,-1,0
  4614.4    0.13       0  4746.4    0.07       0  4945.2    0.13       0
  4993.0    0.05       0  5007.0    0.13       0  5151.5    0.07       0
  5266.2    0.13       0
Bank Sta=4993,5007
XS Rating Curve= 0
Exp/Cntr=0.3,0.1

Type RM Length L Ch R = 1,36832,539,539,539
BEGIN DESCRIPTION:
Grassy Creek 66.0
END DESCRIPTION:
XS GIS Cut Line= 4
      1571989.27       939215.71      1571821.02       939151.89
      1571351.16       939308.51      1570660.91       939610.13
#Sta/Elev= 30
  4665.2  993.34  4686.3  991.69  4837.0  963.90  4845.2  963.17  4873.0  953.71
  4904.1  939.27  4922.1  928.55  4936.6  921.79  4961.0  915.48  4993.0  912.68
  4996.5  907.68  5003.5  907.68  5007.0  912.68  5049.6  914.53  5153.6  917.73
  5163.6  920.74  5175.0  922.29  5186.2  926.73  5196.1  927.80  5212.5  925.45
  5228.8  926.19  5263.4  930.06  5290.7  935.01  5501.4  960.45  5592.8  964.11
  5697.0  964.95  5836.1  970.30  6001.1  980.93  6070.4  987.53  6093.7  987.81
#Mann=7,-1,0
  4665.2     0.1       0  4837.0    0.13       0  4993.0    0.05       0
  5007.0    0.13       0  5049.6    0.07       0  5163.6    0.13       0
  5228.8    0.07       0
Bank Sta=4993,5007
XS Rating Curve= 0
Exp/Cntr=0.3,0.1

Type RM Length L Ch R = 1,36293,584,584,584
BEGIN DESCRIPTION:
Grassy Creek 65.0
END DESCRIPTION:
XS GIS Cut Line= 4
      1571862.45       938570.39      1571646.18       938672.68
      1571234.05       938859.74      1570962.20       938909.44
#Sta/Elev= 30
  4702.4  974.44  4725.0  971.84  4747.6  971.10  4829.9  957.05  4858.8  949.36
  4900.4  933.37  4905.7  933.11  4912.7  930.30  4920.7  926.48  4952.2  916.73
  4971.6  914.90  4993.0  909.92  4996.5  904.92  5003.5  904.92  5007.0  909.92
  5011.8  910.20  5022.4  914.26  5038.1  912.43  5134.8  913.57  5193.3  911.67
  5209.4  910.98  5242.6  914.43  5287.4  915.62  5325.3  915.44  5337.1  915.14
  5370.2  919.40  5398.7  924.19  5451.3  930.59  5625.6  943.82  5670.6  947.95
#Mann=7,-1,0
  4702.4     0.1       0  4912.7    0.13       0  4993.0    0.05       0
  5007.0    0.13       0  5038.1    0.07       0  5193.3    0.13       0
  5325.3    0.07       0
#XS Ineff=2,0
       0                 5260.00    0.00  926.01
Permanent Ineff=
       F       F
Bank Sta=4993,5007
XS Rating Curve= 0
Exp/Cntr=0.3,0.1

Type RM Length L Ch R = 1,35709,822,822,822
BEGIN DESCRIPTION:
Grassy Creek 64.0
END DESCRIPTION:
XS GIS Cut Line= 4
      1571958.92       938234.25      1571593.57       938152.41
      1571508.80       938137.79      1571213.64       938155.33
#Sta/Elev= 30
  4567.5  959.61  4589.9  956.82  4611.5  955.74  4666.4  948.76  4700.7  943.43
  4724.6  941.45  4749.4  937.25  4796.9  927.61  4799.7  927.58  4818.8  923.87
  4834.0  922.03  4849.4  917.45  4861.6  914.63  4892.3  912.19  4924.1  911.33
  4942.4  911.89  4967.5  908.98  4992.6  906.89  4996.1  901.89  5003.9  901.89
  5007.4  906.89  5017.7  909.11  5023.4  911.27  5062.9  910.91  5083.6  912.99
  5165.4  929.93  5229.0  941.05  5244.8  945.40  5269.4  949.41  5323.6  953.33
#Mann=3,-1,0
  4567.5    0.13       0  4992.6    0.05       0  5007.4    0.13       0
Bank Sta=4992.6,5007.4
XS Rating Curve= 0
Exp/Cntr=0.3,0.1

Type RM Length L Ch R = 1,34887,306,306,306
BEGIN DESCRIPTION:
Grassy Creek 63.0
END DESCRIPTION:
XS GIS Cut Line= 4
      1572070.01       937833.54      1571824.47       937383.40
      1571444.50       937310.33      1571158.02       937319.10
#Sta/Elev= 30
  4419.9  928.34  4457.4  925.89  4604.0  920.21  4656.5  915.35  4689.6  910.71
  4714.2  909.09  4829.0  906.55  4949.1  905.25  4981.9  906.60  4989.2  902.54
  4992.6  901.46  4996.1  896.46  5003.9  896.46  5007.4  901.46  5043.7  904.00
  5057.5  904.24  5201.7  904.48  5228.2  906.19  5243.6  905.71  5254.6  907.23
  5311.3  912.00  5323.1  914.34  5349.4  917.98  5392.3  925.89  5412.3  928.95
  5461.4  933.90  5477.3  937.46  5510.8  942.81  5541.3  944.51  5606.2  952.33
#Mann=7,-1,0
  4419.9    0.07       0  4949.1    0.13       0  4992.6    0.05       0
  5007.4    0.13       0  5057.5    0.07       0  5243.6    0.13       0
  5541.3    0.07       0
Bank Sta=4992.6,5007.4
XS Rating Curve= 0
Exp/Cntr=0.3,0.1

Type RM Length L Ch R = 1,34581,273,273,273
BEGIN DESCRIPTION:
Grass Creek 62.7
END DESCRIPTION:
XS GIS Cut Line= 4
      1572301.64       937199.40      1571965.76       937116.08
      1571596.05       937006.73      1571377.39       936998.92
#Sta/Elev= 30
  4504.1  939.01  4553.8  934.77  4640.2  924.80  4694.0  916.77  4714.5  909.28
  4742.0  905.21  4746.9  903.50  4759.7  901.03  4768.1  903.26  4777.0  906.03
  4887.3  904.87  4955.0  902.96  4981.9  901.28  4993.6  899.38  4996.6  894.38
  5003.4  894.38  5006.4  899.38  5018.8  900.05  5023.1  903.64  5028.0  903.78
  5150.1  902.40  5176.7  913.36  5190.3  912.49  5260.9  916.39  5320.5  921.60
  5340.9  929.41  5413.3  944.29  5420.7  944.57  5441.5  949.53  5454.5  950.89
#Mann=5,-1,0
  4504.1    0.15       0  4746.9   0.055       0  4768.1    0.15       0
  4993.6   0.055       0  5006.4    0.15       0
#XS Ineff=1,-1
 4680.00 4777.90  908.22
Permanent Ineff=
       F
Bank Sta=4993.6,5006.4
XS Rating Curve= 0
Exp/Cntr=0.3,0.1

Type RM Length L Ch R = 1,34308,204,204,204
BEGIN DESCRIPTION:
Grassy Creek 62.5
END DESCRIPTION:
XS GIS Cut Line= 5
      1572400.30       936837.99      1571999.85       936858.45
      1571888.78       936811.69      1571719.25       936829.22
      1571356.80       936899.38
#Sta/Elev= 30
  4434.7  948.89  4497.2  941.76  4545.0  937.76  4602.7  929.43  4656.7  918.58
  4682.2  911.02  4716.4  904.86  4726.2  905.29  4790.1  902.14  4817.3  902.21
  4830.7  903.25  4937.6  902.81  4960.2  903.54  4991.2  897.68  4994.2  892.68
  5005.8  892.68  5008.8  897.68  5031.7  898.70  5039.5  900.21  5049.5  898.87
  5083.9  898.17  5099.2  901.34  5105.5  903.73  5119.5  905.65  5147.8  906.00
  5190.8  910.24  5222.1  911.95  5325.3  915.38  5361.4  917.85  5495.8  943.31
#Mann=5,-1,0
  4434.7    0.15       0  4991.2   0.055       0  5008.8    0.15       0
  5119.5    0.08       0  5325.3    0.15       0
#XS Ineff=2,0
    0.00 4958.10  909.84               0
Permanent Ineff=
       F       F
Bank Sta=4991.2,5008.8
XS Rating Curve= 0
Exp/Cntr=0.3,0.1

Type RM Length L Ch R = 1,34104,583,583,583
BEGIN DESCRIPTION:
Grassy Creek 62.0
END DESCRIPTION:
XS GIS Cut Line= 4
      1572309.71       936639.23      1572137.22       936674.31
      1571763.09       936615.85      1571140.54       936706.46
#Sta/Elev= 30
  4532.9  951.29  4563.0  947.52  4595.2  945.28  4638.2  939.32  4675.0  936.50
  4708.9  931.37  4753.8  920.54  4791.5  907.02  4809.3  902.08  4819.9  900.95
  4847.9  901.71  4898.1  902.37  4911.3  901.85  4937.4  898.28  4976.0  895.95
  4991.2  896.60  4994.2  891.60  5005.8  891.60  5008.8  896.60  5020.0  898.94
  5033.8  900.94  5074.4  902.16  5125.1  905.29  5150.9  908.04  5295.8  911.22
  5428.5  917.57  5444.6  918.16  5506.6  926.64  5620.3  938.30  5716.7  951.65
#Mann=8,-1,0
  4532.9    0.13       0  4819.9    0.07       0  4847.9    0.13       0
  4991.2    0.05       0  5008.8    0.13       0  5020.0    0.07       0
  5428.5    0.13       0  5506.6    0.07       0
#XS Ineff=2,0
    0.00 4903.10  907.85               0
Permanent Ineff=
       F       F
Bank Sta=4991.2,5008.8
XS Rating Curve= 0
Exp/Cntr=0.3,0.1

Type RM Length L Ch R = 1,33521,250,250,250
BEGIN DESCRIPTION:
Grassy Creek 61.0
END DESCRIPTION:
XS GIS Cut Line= 4
      1572395.24       936239.91      1572140.05       936106.52
      1571310.55       936286.34      1570939.35       936442.94
#Sta/Elev= 30
  4420.2  969.12  4515.0  964.32  4525.2  964.31  4614.8  957.42  4674.6  947.12
  4695.2  942.68  4722.3  935.18  4737.7  928.95  4787.4  904.91  4793.7  902.81
  4811.4  899.53  4837.8  899.21  4963.1  898.43  4975.8  900.11  4988.9  896.32
  4991.2  894.44  4994.2  889.44  5005.8  889.44  5008.8  894.44  5037.4  898.74
  5066.6  897.80  5092.8  897.81  5199.2  901.11  5309.9  907.33  5457.2  912.30
  5562.9  923.03  5707.3  935.34  5752.2  941.60  5845.7  951.53  5959.8  959.72
#Mann=7,-1,0
  4420.2    0.07       0  4515.0    0.13       0  4837.8    0.07       0
  4963.1    0.13       0  4991.2    0.05       0  5008.8    0.13       0
  5066.6    0.07       0
Bank Sta=4991.2,5008.8
XS Rating Curve= 0
Exp/Cntr=0.3,0.1

Type RM Length L Ch R = 1,33271,337,337,337
BEGIN DESCRIPTION:
Grassy Creek 60.5
END DESCRIPTION:
XS GIS Cut Line= 5
      1572239.49       936066.33      1572040.77       935890.98
      1571842.01       935899.75      1571555.57       936063.43
      1571196.07       936235.87
#Sta/Elev= 30
  4479.6  949.86  4511.2  946.47  4613.5  930.13  4646.7  926.37  4758.0  903.42
  4809.7  900.44  4862.8  899.02  4889.9  899.46  4940.7  897.89  4981.3  899.29
  4984.8  898.86  4991.2  894.22  4994.2  889.22  5005.8  889.22  5008.8  894.22
  5019.3  896.94  5078.8  897.53  5115.1  896.46  5132.8  897.25  5202.9  896.66
  5283.1  899.52  5375.7  904.57  5411.7  907.30  5451.5  911.74  5530.3  922.48
  5579.0  924.79  5593.2  927.58  5624.5  931.05  5654.9  934.13  5672.2  934.99
#Mann=4,-1,0
  4479.6    0.13       0  4991.2    0.05       0  5008.8    0.13       0
  5078.8    0.07       0
Bank Sta=4991.2,5008.8
XS Rating Curve= 0
Exp/Cntr=0.3,0.1

Type RM Length L Ch R = 1,32934,481,481,481
BEGIN DESCRIPTION:
Grassy Creek 60.0
END DESCRIPTION:
XS GIS Cut Line= 4
      1571733.86       935543.16      1571599.41       935657.15
      1571348.04       935882.21      1571035.28       936124.83
#Sta/Elev= 30
  4775.5  960.78  4814.1  950.96  4857.1  936.59  4890.3  927.02  4936.7  910.91
  4970.3  898.23  4991.2  892.40  4994.2  887.40  5005.8  887.40  5008.8  892.40
  5016.9  892.22  5033.2  895.08  5050.0  894.15  5104.1  894.85  5136.6  896.00
  5319.8  896.75  5371.6  899.37  5403.4  904.19  5417.8  908.15  5440.5  911.31
  5456.0  912.52  5541.0  921.94  5577.2  926.57  5597.6  931.38  5609.7  935.06
  5618.5  936.15  5629.0  938.87  5645.4  939.41  5661.4  941.80  5685.0  943.97
#Mann=6,-1,0
  4775.5    0.13       0  4991.2    0.05       0  5008.8    0.13       0
  5136.6    0.07       0  5371.6    0.13       0  5541.0    0.07       0
Bank Sta=4991.2,5008.8
XS Rating Curve= 0
Exp/Cntr=0.3,0.1

Type RM Length L Ch R = 1,32453,430,430,430
BEGIN DESCRIPTION:
Grassy Creek 59.0
END DESCRIPTION:
XS GIS Cut Line= 4
      1571501.94       935242.23      1571258.35       935340.83
      1571101.73       935532.25      1571003.10       935741.11
#Sta/Elev= 30
  4623.5  981.33  4636.3  979.63  4664.8  973.05  4715.9  959.93  4738.2  955.10
  4757.1  951.35  4817.1  941.84  4854.4  935.09  4869.7  931.43  4888.8  925.75
  4917.1  913.78  4935.7  902.49  4944.3  895.36  4962.1  894.00  4979.6  894.26
  4991.2  890.23  4994.2  885.23  5005.8  885.23  5008.8  890.23  5029.1  890.38
  5032.4  890.41  5048.9  894.59  5082.9  906.68  5132.4  922.32  5168.5  932.19
  5196.0  938.29  5257.6  946.90  5290.6  950.71  5314.2  953.08  5364.6  956.52
#Mann=5,-1,0
  4623.5    0.13       0  4991.2    0.05       0  5008.8    0.13       0
  5029.1    0.07       0  5048.9    0.13       0
Bank Sta=4991.2,5008.8
XS Rating Curve= 0
Exp/Cntr=0.3,0.1

Type RM Length L Ch R = 1,32023,374,374,374
BEGIN DESCRIPTION:
Grassy Creek 58.0
END DESCRIPTION:
XS GIS Cut Line= 3
      1570979.94       934963.74      1570678.28       935456.84
      1570817.47       935688.83
#Sta/Elev= 30
  4678.5  976.20  4701.8  967.03  4750.1  950.26  4812.2  925.07  4837.4  913.94
  4853.2  907.72  4872.9  901.53  4905.1  894.25  4924.9  892.43  4936.7  893.17
  4955.1  889.24  4971.9  887.72  4991.2  887.85  4994.2  882.85  5005.8  882.85
  5008.8  887.85  5024.3  892.02  5035.5  892.40  5096.8  892.89  5127.5  894.73
  5148.5  896.89  5173.0  901.32  5193.3  906.54  5233.4  918.81  5281.5  928.23
  5353.3  937.38  5398.6  944.76  5439.7  949.93  5484.0  954.55  5527.1  956.72
#Mann=5,-1,0
  4678.5    0.13       0  4991.2    0.05       0  5008.8    0.13       0
  5035.5    0.07       0  5193.3    0.13       0
Bank Sta=4991.2,5008.8
XS Rating Curve= 0
Exp/Cntr=0.3,0.1

Type RM Length L Ch R = 1,31649,414,414,414
BEGIN DESCRIPTION:
Grassy Creek 57.5
END DESCRIPTION:
XS GIS Cut Line= 4
      1570515.02       934911.79      1570550.10       935291.79
      1570585.17       935499.32      1570754.74       935633.80
#Sta/Elev= 30
  4884.3  939.68  4896.5  935.59  4921.5  924.34  4932.5  918.64  4948.6  908.35
  4964.2  897.24  4974.8  891.09  4991.2  885.26  4994.2  880.26  5005.8  880.26
  5008.8  885.26  5033.8  887.39  5038.0  889.89  5054.2  890.68  5073.3  892.54
  5124.1  895.57  5141.0  895.95  5196.7  898.47  5264.7  900.09  5319.5  902.98
  5355.0  907.46  5415.6  917.06  5469.4  923.27  5491.9  926.78  5498.3  927.25
  5524.3  930.01  5565.3  935.35  5587.1  937.71  5595.4  937.93  5692.8  949.74
#Mann=5,-1,0
  4884.3    0.13       0  4991.2    0.05       0  5008.8    0.13       0
  5073.3    0.07       0  5498.3    0.13       0
Bank Sta=4991.2,5008.8
XS Rating Curve= 0
Exp/Cntr=0.3,0.1

Type RM Length L Ch R = 1,31235,531,531,531
BEGIN DESCRIPTION:
Grassy Creek 57.0
END DESCRIPTION:
XS GIS Cut Line= 4
      1570341.84       935015.99      1570185.22       935242.21
      1570475.25       935532.25      1570863.88       935717.86
#Sta/Elev= 30
  4612.4  935.92  4689.0  930.48  4715.7  926.41  4788.0  917.70  4828.3  911.23
  4832.9  912.81  4871.9  912.00  4879.6  910.89  4895.7  907.00  4955.0  883.96
  4965.9  884.01  4980.0  882.00  4991.2  882.21  4994.2  877.21  5005.8  877.21
  5008.8  882.21  5030.0  884.27  5084.8  894.29  5101.4  896.28  5130.0  897.32
  5162.5  903.89  5234.4  910.52  5380.6  928.10  5479.4  937.05  5495.1  939.47
  5521.7  941.04  5530.2  942.83  5540.4  942.78  5629.0  953.73  5728.4  959.03
#Mann=6,-1,0
  4612.4    0.07       0  4715.7    0.13       0  4991.2    0.05       0
  5008.8    0.13       0  5030.0    0.07       0  5380.6    0.13       0
Bank Sta=4991.2,5008.8
XS Rating Curve= 0
Exp/Cntr=0.3,0.1

Type RM Length L Ch R = 1,30704,471,471,471
BEGIN DESCRIPTION:
Grassy Creek 56.0
END DESCRIPTION:
XS GIS Cut Line= 4
      1570278.93       935091.94      1569897.97       935490.48
      1569862.24       935902.68      1569731.19       936008.16
#Sta/Elev= 30
  4289.9  927.23  4487.6  906.13  4543.8  900.57  4617.5  894.54  4638.5  890.63
  4669.1  889.35  4679.3  887.86  4859.4  882.63  4932.7  882.19  4963.0  881.16
  4976.4  881.94  4979.8  881.21  4990.9  879.91  4993.9  874.91  5006.1  874.91
  5009.1  879.91  5028.9  881.75  5047.6  881.95  5081.6  880.73  5093.9  881.57
  5108.2  887.52  5121.7  894.83  5163.7  914.10  5178.4  919.03  5220.5  929.69
  5242.6  931.86  5308.1  930.32  5329.4  933.17  5383.9  942.22  5423.2  946.54
#Mann=4,-1,0
  4289.9    0.07       0  4979.8    0.13       0  4990.9    0.05       0
  5009.1    0.13       0
Bank Sta=4990.9,5009.1
XS Rating Curve= 0
Exp/Cntr=0.5,0.3

Type RM Length L Ch R = 1,30233,94,94,94
BEGIN DESCRIPTION:
Mt Zion Rd (GC) us
END DESCRIPTION:
XS GIS Cut Line= 6
      1570298.64       935055.37      1569812.69       935538.52
      1569635.73       935572.22      1569208.79       935473.91
      1569107.67       935490.76      1569012.18       935589.06
#Sta/Elev= 30
  3994.9  930.85  4034.3  927.33  4267.9  902.54  4362.0  894.92  4393.9  893.32
  4404.9  891.75  4431.6  890.64  4449.6  888.60  4481.3  888.12  4597.7  883.46
  4676.4  881.78  4715.3  881.22  4809.1  881.70  4910.3  879.84  4949.8  880.31
  4966.5  877.29  4983.5  876.10  4992.0  871.40  5008.0  871.40  5016.5  876.10
  5024.9  879.03  5032.4  881.24  5062.1  879.80  5074.9  880.41  5120.4  879.73
  5203.6  880.63  5210.1  881.65  5270.2  885.29  5403.6  900.19  5540.6  916.67
#Mann=5,-1,0
  3994.9    0.07       0  4910.3    0.13       0  4983.5    0.05       0
  5016.5    0.13       0  5024.9    0.07       0
#XS Ineff=2,0
    0.00 4942.00  883.17 5058.00    0.00  883.57
Permanent Ineff=
       F       F
Bank Sta=4983.5,5016.5
XS Rating Curve= 0
Exp/Cntr=0.5,0.3

Type RM Length L Ch R =3,30190,,,
BEGIN DESCRIPTION:
Mt Zion Rd (GC) TOR
Structure ID: LDS_GC_05
Approximate Survey Structure
END DESCRIPTION:
Bridge Culvert--1,0,-1,-1,0
Deck Dist Width WeirC Skew NumUp NumDn MinLoCord MaxHiCord MaxSubmerge Is_Ogee
30.5,25,3,,17,17,,,0.95,0,1,1,,,
  3987.4  4252.2  4390.8  4538.3  4665.5  4796.3  4851.2  4972.5  4972.5  5027.5
  5027.5  5131.9  5239.4  5329.7  5440.6  5534.6  5594.2
  933.51  906.85  894.66  888.24  884.29  882.76  883.17  882.70  882.70  882.70
  882.70  883.90  885.95  888.48  900.91  914.18  918.96
  851.40  851.40  851.40  851.40  851.40  851.40  851.40  851.40  880.70  880.70
  851.40  851.40  851.40  851.40  851.40  851.40  851.40
  3987.4  4252.2  4390.8  4538.3  4665.5  4796.3  4851.2  4972.5  4972.5  5027.5
  5027.5  5131.9  5239.4  5329.7  5440.6  5534.6  5594.2
  933.51  906.85  894.66  888.24  884.29  882.76  883.17  882.70  882.70  882.70
  882.70  883.90  885.95  888.48  900.91  914.18  918.96
  851.40  851.40  851.40  851.40  851.40  851.40  851.40  851.40  880.70  880.70
  851.40  851.40  851.40  851.40  851.40  851.40  851.40
Pier Skew, UpSta & Num, DnSta & Num=,5000,2,5000,2,0,0,0,0,0
       2       2
  871.40  880.70
       2       2
  871.15  880.70
BR Coef=1,1,0,1.25,0,,,0.8,0,2,0,
WSPro=,,,, 1 ,,,, 0 ,,,, 0 ,,,,-1 ,-1 ,-1 , 0 , 0 , 0 , 0 , 0
BC Design=,,0,,0,,,,,,

Type RM Length L Ch R = 1,30139,624,624,624
BEGIN DESCRIPTION:
Mt Zion Rd (GC) ds
END DESCRIPTION:
XS GIS Cut Line= 6
      1570250.89       935041.33      1569809.88       935457.06
      1569680.68       935487.96      1569203.17       935384.03
      1569065.53       935420.54      1568986.89       935555.36
#Sta/Elev= 30
  4072.5  930.92  4104.5  928.65  4160.8  923.07  4211.7  916.93  4332.8  899.34
  4367.1  897.72  4391.3  894.08  4617.9  886.67  4639.3  884.52  4733.5  880.63
  4880.0  878.97  4923.0  879.21  4932.8  879.36  4983.5  875.85  4992.0  871.15
  5008.0  871.15  5016.5  875.85  5026.0  876.65  5043.9  878.16  5072.2  877.38
  5207.2  878.34  5251.6  881.39  5282.1  885.81  5302.6  886.82  5328.2  889.44
  5418.1  891.50  5439.9  895.25  5472.9  898.89  5577.9  914.92  5600.3  915.90
#Mann=5,-1,0
  4072.5    0.07       0  4923.0    0.13       0  4983.5    0.05       0
  5016.5    0.13       0  5026.0    0.07       0
#XS Ineff=2,0
    0.00 4934.00  883.30 5066.00    0.00  883.26
Permanent Ineff=
       F       F
Bank Sta=4983.5,5016.5
XS Rating Curve= 0
Exp/Cntr=0.5,0.3

Type RM Length L Ch R = 1,29515,437,437,437
BEGIN DESCRIPTION:
Grassy Creek 55.0
END DESCRIPTION:
XS GIS Cut Line= 5
      1569860.39       934662.13      1569616.75       934853.57
      1569100.49       935126.20      1568972.87       935364.03
      1568970.03       935583.42
#Sta/Elev= 30
  4472.0  942.12  4492.9  939.41  4563.3  920.70  4612.5  910.80  4635.9  903.91
  4661.5  903.78  4754.7  894.39  4771.7  889.85  4792.0  878.24  4800.8  874.69
  4813.1  875.97  4875.4  875.59  4945.7  876.15  4968.4  876.35  4990.5  872.79
  4993.5  867.79  5006.5  867.79  5009.5  872.79  5010.3  875.49  5015.0  876.02
  5178.5  874.79  5245.7  876.12  5349.9  889.77  5457.6  897.86  5568.3  898.47
  5624.0  895.78  5656.5  896.18  5684.6  898.61  5763.6  909.31  5855.0  918.18
#Mann=6,-1,0
  4472.0    0.13       0  4875.4    0.07       0  4945.7    0.13       0
  4990.5    0.05       0  5009.5    0.13       0  5015.0    0.07       0
Bank Sta=4990.5,5009.5
XS Rating Curve= 0
Exp/Cntr=0.3,0.1

Type RM Length L Ch R = 1,29078,448,448,448
BEGIN DESCRIPTION:
Grassy Creek 54.0
END DESCRIPTION:
XS GIS Cut Line= 3
      1569599.32       934476.53      1569286.11       934621.54
      1568613.19       934992.81
#Sta/Elev= 30
  4495.2  938.31  4542.6  929.82  4554.8  929.54  4569.0  926.99  4605.2  925.24
  4644.5  921.47  4827.6  900.36  4854.4  893.60  4882.7  880.97  4898.2  875.15
  4910.5  873.63  4922.0  873.99  4938.3  871.73  4955.0  871.32  4976.0  872.31
  4990.5  870.84  4993.5  865.84  5006.5  865.84  5009.5  870.84  5027.2  874.13
  5038.8  873.98  5136.7  872.50  5169.1  873.35  5190.1  877.09  5245.9  890.76
  5325.3  901.79  5351.0  903.97  5452.2  918.24  5567.3  930.67  5608.9  936.13
#Mann=5,-1,0
  4495.2    0.13       0  4990.5    0.05       0  5009.5    0.13       0
  5038.8    0.13       0  5452.2    0.07       0
Bank Sta=4990.5,5009.5
XS Rating Curve= 0
Exp/Cntr=0.3,0.1

Type RM Length L Ch R = 1,28630,356,356,356
BEGIN DESCRIPTION:
Grassy Creek 53.7
END DESCRIPTION:
XS GIS Cut Line= 4
      1569293.25       934298.02      1569164.66       934327.24
      1568936.67       934435.39      1568711.64       934613.66
#Sta/Elev= 30
  4484.7  917.45  4508.9  912.87  4532.8  905.79  4553.4  897.68  4562.9  894.60
  4573.3  889.92  4586.8  886.17  4601.0  882.50  4618.8  879.43  4650.1  876.61
  4751.8  872.05  4766.3  871.05  4780.7  871.19  4803.6  871.64  4831.6  870.75
  4904.8  872.10  4923.9  871.07  4937.9  872.12  4954.2  871.58  4970.5  869.18
  4990.5  868.42  4993.5  863.42  5006.5  863.42  5009.5  868.42  5023.6  869.86
  5033.8  872.88  5086.5  895.62  5113.6  905.25  5139.7  912.71  5156.0  914.96
#Mann=7,-1,0
  4484.7    0.13       0  4586.8    0.07       0  4751.8    0.13       0
  4780.7    0.07       0  4904.8    0.13       0  4990.5    0.05       0
  5009.5    0.13       0
Bank Sta=4990.5,5009.5
XS Rating Curve= 0
Exp/Cntr=0.3,0.1

Type RM Length L Ch R = 1,28274,145,145,145
BEGIN DESCRIPTION:
Grassy Creek 53.5
END DESCRIPTION:
XS GIS Cut Line= 6
      1568927.91       933920.96      1568772.99       934105.10
      1568708.69       934181.10      1568626.85       934233.71
      1568597.62       934306.78      1568480.69       934502.64
#Sta/Elev= 30
  4602.9  929.35  4634.6  926.69  4669.2  921.99  4704.4  913.44  4738.8  902.18
  4793.4  877.26  4810.7  872.96  4833.3  870.63  4845.2  868.60  4879.4  869.52
  4912.9  867.32  4946.5  869.37  4965.9  867.31  4990.5  865.96  4993.5  860.96
  5006.5  860.96  5009.5  865.96  5016.6  865.94  5025.1  868.80  5037.5  869.39
  5083.6  869.14  5129.0  869.61  5143.0  870.42  5158.5  869.98  5175.1  872.23
  5207.2  884.97  5229.8  891.62  5305.9  901.58  5330.6  903.36  5347.2  903.74
#Mann=3,-1,0
  4602.9    0.13       0  4990.5    0.05       0  5009.5    0.13       0
Bank Sta=4990.5,5009.5
XS Rating Curve= 0
Exp/Cntr=0.3,0.1

Type RM Length L Ch R = 1,28129,826,826,826
BEGIN DESCRIPTION:
Grassy Creek 53.0
END DESCRIPTION:
XS GIS Cut Line= 3
      1569036.68       933768.84      1568305.79       934302.50
      1568004.13       934575.15
#Sta/Elev= 30
  4477.5  951.65  4593.6  941.35  4743.7  919.98  4827.9  896.93  4869.6  878.11
  4890.2  871.34  4916.9  867.13  4955.1  866.36  4968.6  867.79  4990.3  865.53
  4990.5  864.51  4993.5  859.51  5006.5  859.51  5009.5  864.51  5038.7  868.78
  5090.2  866.88  5130.9  865.77  5198.6  866.49  5214.0  867.90  5242.8  873.66
  5303.9  902.09  5333.0  909.56  5365.3  914.33  5404.3  916.52  5496.2  917.46
  5546.6  920.88  5598.7  922.49  5718.9  924.07  5732.0  925.48  5789.1  928.15
#Mann=6,-1,0
  4477.5    0.13       0  4990.5    0.05       0  5009.5    0.13       0
  5090.2    0.07       0  5214.0    0.13       0  5732.0    0.07       0
Bank Sta=4990.5,5009.5
XS Rating Curve= 0
Exp/Cntr=0.3,0.1

Type RM Length L Ch R = 1,27303,584,584,584
BEGIN DESCRIPTION:
Grassy Creek 52.0
END DESCRIPTION:
XS GIS Cut Line= 4
      1568561.05       933084.32      1568427.60       933235.17
      1567835.93       933832.64      1567841.73       934261.93
#Sta/Elev= 30
  4445.5  945.38  4474.3  936.81  4559.0  916.43  4613.5  889.07  4625.9  885.09
  4649.9  868.64  4753.2  864.47  4912.3  862.16  4945.5  863.02  4965.8  864.18
  4990.4  861.02  4993.4  856.02  5006.6  856.02  5009.6  861.02  5050.1  864.50
  5083.9  863.12  5135.3  863.67  5241.0  869.10  5288.3  869.82  5480.0  880.58
  5518.9  885.78  5547.3  887.75  5556.4  890.55  5658.1  906.72  5689.9  910.77
  5705.2  910.75  5721.3  914.04  5750.2  915.99  5784.0  920.91  5917.1  925.92
#Mann=6,-1,0
  4445.5    0.13       0  4753.2    0.07       0  4945.5    0.13       0
  4990.4    0.05       0  5009.6    0.13       0  5083.9    0.07       0
#XS Ineff=2,0
    0.00 4731.90  879.93               0
Permanent Ineff=
       F       F
Bank Sta=4990.4,5009.6
XS Rating Curve= 0
Exp/Cntr=0.3,0.1

Type RM Length L Ch R = 1,26719,508,508,508
BEGIN DESCRIPTION:
Grassy Creek 51.0
END DESCRIPTION:
XS GIS Cut Line= 5
      1568125.99       932904.52      1567834.75       933011.95
      1567805.52       933090.87      1567720.76       933394.85
      1567484.02       933678.35
#Sta/Elev= 30
  4519.8  947.68  4597.9  940.63  4634.5  934.45  4664.8  928.13  4693.8  919.30
  4736.7  900.18  4770.9  886.52  4806.4  870.54  4819.2  866.24  4835.0  863.13
  4853.4  862.08  4940.3  863.41  4983.6  860.80  4990.4  859.28  4993.4  854.28
  5006.6  854.28  5009.6  859.28  5045.3  858.87  5060.5  861.07  5084.8  862.58
  5101.2  861.78  5136.7  863.04  5188.5  862.68  5237.9  865.18  5253.1  866.10
  5319.0  866.63  5407.1  872.78  5458.5  878.03  5524.1  889.07  5599.3  899.91
#Mann=5,-1,0
  4519.8    0.13       0  4990.4    0.05       0  5009.6    0.13       0
  5237.9    0.07       0  5524.1    0.13       0
#XS Ineff=2,0
    0.00 4930.20  873.08 5099.60    0.00  873.08
Permanent Ineff=
       F       F
Bank Sta=4990.4,5009.6
XS Rating Curve= 0
Exp/Cntr=0.3,0.1

Type RM Length L Ch R = 1,26211,653,653,653
BEGIN DESCRIPTION:
Grassy Creek 50.0
END DESCRIPTION:
XS GIS Cut Line= 5
      1567296.47       932614.47      1567296.47       932881.33
      1567354.47       933142.36      1567337.07       933478.80
      1567174.68       933641.19
#Sta/Elev= 30
  4554.8  914.74  4610.6  910.93  4647.2  907.37  4763.0  900.49  4806.4  896.47
  4852.7  889.55  4870.7  885.61  4932.0  874.62  4950.4  869.51  4990.4  855.74
  4993.4  850.74  5006.6  850.74  5009.6  855.74  5026.0  859.35  5032.0  861.63
  5046.5  860.11  5074.3  858.67  5109.6  858.35  5230.8  858.23  5275.3  859.12
  5310.0  859.99  5317.1  860.73  5356.7  872.72  5382.1  878.75  5421.7  890.78
  5457.3  899.83  5505.3  910.09  5590.7  922.49  5635.2  925.84  5655.6  925.74
#Mann=5,-1,0
  4554.8    0.13       0  4990.4    0.05       0  5009.6    0.13       0
  5109.6    0.07       0  5275.3    0.13       0
Bank Sta=4990.4,5009.6
XS Rating Curve= 0
Exp/Cntr=0.3,0.1

Type RM Length L Ch R = 1,25558,413,413,413
BEGIN DESCRIPTION:
Grassy Creek 49.0
END DESCRIPTION:
XS GIS Cut Line= 5
      1567197.88       932492.66      1566867.22       932840.72
      1566774.40       933008.94      1566820.81       933177.16
      1567047.03       933525.19
#Sta/Elev= 30
  4424.8  914.51  4464.8  911.29  4585.7  897.84  4643.3  892.65  4667.9  889.02
  4753.5  883.77  4821.3  881.79  4855.2  879.61  4888.3  876.05  4923.4  871.02
  4971.7  855.37  4990.4  853.00  4993.4  848.00  5006.6  848.00  5009.6  853.00
  5058.0  861.68  5110.3  873.20  5172.3  881.35  5198.7  883.01  5214.8  881.30
  5313.5  888.33  5358.5  897.26  5409.8  899.30  5428.2  902.33  5436.9  901.77
  5458.9  904.28  5519.5  908.12  5601.1  908.46  5637.4  912.53  5686.6  916.25
#Mann=3,-1,0
  4424.8    0.13       0  4990.4    0.05       0  5009.6    0.13       0
Bank Sta=4990.4,5009.6
XS Rating Curve= 0
Exp/Cntr=0.3,0.1

Type RM Length L Ch R = 1,25145,334,334,334
BEGIN DESCRIPTION:
Grassy Creek 48.0
END DESCRIPTION:
XS GIS Cut Line= 4
      1566960.03       932434.67      1566414.76       932771.12
      1566281.35       933061.15      1566327.75       933217.75
#Sta/Elev= 30
  4455.6  906.66  4472.2  906.72  4487.8  904.75  4516.5  903.18  4584.5  896.34
  4634.4  889.16  4741.0  869.43  4783.6  862.38  4843.4  856.53  4925.7  853.18
  4970.0  853.86  4989.7  850.61  4992.7  845.61  5007.3  845.61  5010.3  850.61
  5026.3  855.63  5043.4  858.49  5060.9  862.71  5180.1  875.76  5254.6  881.46
  5266.2  883.08  5295.3  883.86  5337.6  888.82  5353.3  889.89  5363.5  892.38
  5400.6  896.16  5468.0  899.13  5485.8  900.34  5552.1  907.58  5578.9  908.11
#Mann=5,-1,0
  4455.6    0.13       0  4783.6    0.07       0  4970.0    0.13       0
  4989.7    0.05       0  5010.3    0.13       0
Bank Sta=4989.7,5010.3
XS Rating Curve= 0
Exp/Cntr=0.3,0.1

Type RM Length L Ch R = 1,24811,488,488,488
BEGIN DESCRIPTION:
Grassy Creek 47.0
END DESCRIPTION:
XS GIS Cut Line= 4
      1566234.93       932376.64      1566339.35       932794.32
      1566269.74       933055.35      1566327.76       933241.01
#Sta/Elev= 30
  4790.0  930.20  4852.8  917.45  4886.4  904.96  4892.2  902.49  4908.9  892.54
  4938.9  879.38  4978.4  853.15  4989.7  848.34  4992.7  843.34  5007.3  843.34
  5010.3  848.34  5021.2  850.01  5030.7  853.03  5040.6  852.06  5047.1  851.35
  5093.7  853.44  5105.1  852.92  5136.9  854.76  5241.5  873.23  5276.3  877.58
  5288.0  877.97  5302.0  880.31  5313.4  880.84  5329.9  883.55  5412.6  891.88
  5490.7  897.52  5550.0  899.09  5633.2  906.85  5663.9  907.85  5685.2  907.12
#Mann=5,-1,0
  4790.0    0.13       0  4989.7    0.05       0  5010.3    0.13       0
  5040.6    0.07       0  5136.9    0.13       0
Bank Sta=4989.7,5010.3
XS Rating Curve= 0
Exp/Cntr=0.3,0.1

Type RM Length L Ch R = 1,24323,961,961,961
BEGIN DESCRIPTION:
Grassy Creek 46.0
END DESCRIPTION:
XS GIS Cut Line= 2
      1565834.69       932341.89      1565840.49       933385.98
#Sta/Elev= 30
  4646.7  917.84  4668.1  915.60  4713.3  908.67  4726.2  904.23  4768.3  892.98
  4782.5  887.14  4796.6  883.71  4825.7  869.59  4840.8  860.78  4858.6  853.74
  4879.0  850.02  4896.0  849.14  4980.7  850.16  4989.7  845.69  4992.7  840.69
  5007.3  840.69  5010.3  845.69  5035.5  848.80  5043.9  851.09  5083.3  850.91
  5107.4  849.03  5173.7  849.59  5212.3  851.28  5261.0  865.34  5299.6  874.34
  5382.1  888.32  5432.4  895.52  5556.1  907.64  5634.1  911.26  5690.8  917.35
#Mann=7,-1,0
  4646.7    0.13       0  4668.1    0.15       0  4858.6    0.13       0
  4989.7    0.05       0  5010.3    0.13       0  5107.4    0.07       0
  5212.3    0.13       0
Bank Sta=4989.7,5010.3
XS Rating Curve= 0
Exp/Cntr=0.3,0.1

Type RM Length L Ch R = 1,23362,917,917,917
BEGIN DESCRIPTION:
Grassy Creek 45.0
END DESCRIPTION:
XS GIS Cut Line= 4
      1565794.09       932301.26      1565434.44       932289.66
      1564981.99       932562.29      1564755.77       932852.31
#Sta/Elev= 30
  4203.0  916.65  4219.8  914.97  4260.6  909.82  4295.5  902.18  4311.0  900.33
  4441.4  875.17  4526.0  860.25  4553.5  857.04  4574.8  856.86  4628.1  848.68
  4659.2  846.90  4882.3  845.24  4936.3  843.90  4950.3  842.41  4957.2  844.01
  4976.0  846.98  4989.7  842.13  4992.7  837.13  5007.3  837.13  5010.3  842.13
  5019.3  846.42  5034.2  846.35  5051.1  849.60  5072.2  850.74  5087.8  855.76
  5120.5  860.10  5149.4  866.71  5279.5  887.41  5426.6  904.80  5458.9  907.01
#Mann=6,-1,0
  4203.0    0.13       0  4219.8    0.15       0  4526.0    0.07       0
  4957.2    0.13       0  4989.7    0.05       0  5010.3    0.13       0
Bank Sta=4989.7,5010.3
XS Rating Curve= 0
Exp/Cntr=0.3,0.1

Type RM Length L Ch R = 1,22445,649,649,649
BEGIN DESCRIPTION:
Grassy Creek 44.0
END DESCRIPTION:
XS GIS Cut Line= 4
      1565428.68       931657.38      1564604.94       931715.39
      1564355.51       931692.18      1564053.92       931750.18
#Sta/Elev= 30
  4352.2  920.77  4378.0  920.11  4415.1  915.94  4479.7  905.61  4519.8  896.29
  4574.2  879.68  4624.7  860.13  4660.1  843.40  4687.2  841.83  4898.2  840.71
  4929.2  838.59  4934.7  838.25  4947.8  842.88  4963.3  843.40  4987.3  838.33
  4990.3  833.33  5009.7  833.33  5012.7  838.33  5015.0  840.34  5027.8  843.08
  5038.5  848.41  5053.6  849.87  5123.0  865.62  5189.6  871.28  5312.1  874.97
  5409.3  883.53  5454.7  886.31  5501.6  892.49  5570.4  899.31  5735.6  912.80
#Mann=8,-1,0
  4352.2    0.15       0  4660.1    0.07       0  4929.2    0.13       0
  4987.3    0.05       0  5012.7    0.13       0  5189.6    0.07       0
  5409.3    0.13       0  5501.6    0.07       0
Bank Sta=4987.3,5012.7
XS Rating Curve= 0
Exp/Cntr=0.5,0.3

Type RM Length L Ch R = 1,21796,99,99,99
BEGIN DESCRIPTION:
Stony Ridge Rd (GC) us
END DESCRIPTION:
XS GIS Cut Line= 5
      1565815.18       931141.36      1565433.18       931051.30
      1565169.23       931051.30      1564467.42       931097.88
      1564004.74       931430.14
#Sta/Elev= 30
  3892.9  902.10  4109.9  880.11  4215.4  863.28  4281.9  856.00  4296.7  855.69
  4307.1  853.34  4385.5  847.52  4442.6  844.06  4546.6  841.36  4916.8  837.74
  4961.7  837.33  4973.8  835.44  4978.8  835.90  4990.8  830.50  5009.2  830.50
  5021.2  835.90  5033.6  839.36  5156.9  839.57  5202.3  841.40  5230.4  846.21
  5242.7  850.50  5303.2  856.48  5349.9  863.81  5376.1  865.39  5432.7  865.90
  5488.1  864.82  5517.2  865.76  5555.7  871.21  5692.4  879.65  5822.3  891.29
#Mann=5,-1,0
  3892.9    0.07       0  4916.8    0.13       0  4978.8    0.05       0
  5021.2    0.13       0  5202.3    0.07       0
#XS Ineff=2,0
    0.00 4911.50  845.77 5088.50    0.00  846.25
Permanent Ineff=
       F       F
Bank Sta=4978.8,5021.2
XS Rating Curve= 0
Exp/Cntr=0.5,0.3

Type RM Length L Ch R =3,21745,,,
BEGIN DESCRIPTION:
Stony Ridge Rd (GC) TOR
Structure ID: LDS_GC_04
Approximate Survey Structure
END DESCRIPTION:
Bridge Culvert--1,0,-1,-1,0
Deck Dist Width WeirC Skew NumUp NumDn MinLoCord MaxHiCord MaxSubmerge Is_Ogee
38.5,25,3,,15,15,,,0.95,0,1,1,,,
  3841.5  4025.4  4138.7  4353.3  4447.2  4553.8  4777.8  4950.0  4950.0  5050.0
  5050.0  5133.9  5306.5  5555.8  5941.8
  902.65  885.53  874.35  856.64  851.32  848.06  846.36  845.60  845.60  845.60
  845.60  846.25  852.31  867.38  893.28
  810.50  810.50  810.50  810.50  810.50  810.50  810.50  810.50  843.60  843.60
  810.50  810.50  810.50  810.50  810.50
  3841.5  4025.4  4138.7  4353.3  4447.2  4553.8  4777.8  4950.0  4950.0  5050.0
  5050.0  5133.9  5306.5  5555.8  5941.8
  902.65  885.53  874.35  856.64  851.32  848.06  846.36  845.60  845.60  845.60
  845.60  846.25  852.31  867.38  893.28
  810.50  810.50  810.50  810.50  810.50  810.50  810.50  810.50  843.60  843.60
  810.50  810.50  810.50  810.50  810.50
Pier Skew, UpSta & Num, DnSta & Num=,4975,2,4975,2,0,0,0,0,0
       1       1
  837.16  843.60
       1       1
  836.91  843.60
Pier Skew, UpSta & Num, DnSta & Num=,5025,2,5025,2,0,0,0,0,0
       1       1
  837.16  843.60
       1       1
  836.91  843.60
Abutment Skew #Up #Dn=,2,2
  4950.0  4962.5
  843.60  837.25
  4950.0  4962.5
  843.60  834.07
Abutment Skew #Up #Dn=,2,2
  5037.5  5050.0
  839.35  843.60
  5037.5  5050.0
  835.53  843.60
BR Coef=1,1,0,1.25,0,,,0.8,0,2,0,
WSPro=,,,, 1 ,,,, 0 ,,,, 0 ,,,,-1 ,-1 ,-1 , 0 , 0 , 0 , 0 , 0
BC Design=,,0,,0,,,,,,

Type RM Length L Ch R = 1,21697,245,245,245
BEGIN DESCRIPTION:
Stony Ridge Rd (GC) ds
END DESCRIPTION:
XS GIS Cut Line= 6
      1565849.28       931051.30      1565333.81       930948.82
      1564777.96       930976.77      1564473.63       931007.83
      1564312.16       931069.93      1563896.07       931420.81
#Sta/Elev= 30
  3839.2  903.33  4030.4  883.35  4330.2  844.06  4423.3  840.51  4913.7  836.80
  4978.8  835.65  4990.8  830.25  5009.2  830.25  5021.2  835.65  5096.6  839.00
  5171.6  836.45  5179.4  839.79  5209.1  837.65  5220.6  841.73  5241.1  838.69
  5246.2  842.30  5273.3  845.19  5309.1  845.32  5381.1  851.39  5401.1  852.42
  5413.1  857.89  5430.5  859.13  5587.2  860.42  5613.5  861.29  5651.5  868.91
  5691.3  872.74  5760.5  873.20  5811.1  878.12  5941.8  890.78  5944.6  890.99
#Mann=8,-1,0
  3839.2    0.07       0  4913.7    0.13       0  4978.8    0.05       0
  5021.2    0.13       0  5381.1    0.07       0  5587.2    0.13       0
  5811.1    0.07       0  5941.8    0.13       0
#XS Ineff=2,0
    0.00 4914.50  845.67 5085.50    0.00  846.17
Permanent Ineff=
       F       F
Bank Sta=4978.8,5021.2
XS Rating Curve= 0
Exp/Cntr=0.5,0.3

Type RM Length L Ch R = 1,21452,541,541,541
BEGIN DESCRIPTION:
Grassy Creek 43.5
END DESCRIPTION:
XS GIS Cut Line= 5
      1565800.68       930835.28      1565396.91       930743.92
      1564993.14       930720.34      1564341.82       930764.55
      1564076.52       930788.13
#Sta/Elev= 30
  3869.2  883.12  4026.0  862.66  4127.6  854.53  4206.1  843.91  4260.6  840.22
  4356.9  837.53  4396.1  838.53  4737.8  838.18  4920.1  836.43  4950.1  834.80
  4954.8  834.71  4964.7  837.67  4985.9  834.91  4987.3  833.38  4990.3  828.38
  5009.7  828.38  5012.7  833.38  5060.3  838.04  5098.0  836.98  5135.7  838.95
  5167.4  842.56  5181.8  846.03  5273.1  853.46  5353.0  863.58  5365.8  864.57
  5414.6  863.87  5429.9  867.77  5449.9  869.90  5490.6  871.55  5606.8  880.35
#Mann=5,-1,0
  3869.2    0.07       0  4950.1    0.13       0  4987.3    0.05       0
  5012.7    0.13       0  5060.3    0.07       0
#XS Ineff=2,0
    0.00 4650.10  847.38               0
Permanent Ineff=
       F       F
Bank Sta=4987.3,5012.7
XS Rating Curve= 0
Exp/Cntr=0.3,0.1

Type RM Length L Ch R = 1,20911,521,521,521
BEGIN DESCRIPTION:
Grassy Creek 43.0
END DESCRIPTION:
XS GIS Cut Line= 4
      1566211.76       930665.47      1565620.06       930387.03
      1564459.92       930213.01      1563937.86       930555.25
#Sta/Elev= 30
  3309.8  914.98  3411.3  901.93  3457.5  890.97  3478.1  890.55  3573.7  877.69
  3684.6  868.13  3711.8  864.98  3771.9  861.99  3838.9  853.20  3963.7  842.45
  4063.9  837.77  4223.7  834.46  4523.0  835.50  4908.7  833.82  4938.5  835.05
  4954.5  838.06  4977.1  833.12  4987.3  832.59  4990.3  827.59  5009.7  827.59
  5012.7  832.59  5027.1  836.40  5093.1  835.04  5114.5  846.95  5140.3  856.89
  5225.5  868.36  5252.3  869.53  5332.8  869.62  5461.7  879.07  5761.1  886.35
#Mann=6,-1,0
  3309.8    0.13       0  3684.6    0.07       0  4908.7    0.13       0
  4987.3    0.05       0  5012.7    0.13       0  5252.3    0.07       0
#XS Ineff=2,0
    0.00 4394.80  857.28               0
Permanent Ineff=
       F       F
Bank Sta=4987.3,5012.7
XS Rating Curve= 0
Exp/Cntr=0.3,0.1

Type RM Length L Ch R = 1,20390,972,972,972
BEGIN DESCRIPTION:
Grassy Creek 42.0
END DESCRIPTION:
XS GIS Cut Line= 4
      1566083.85       930260.66      1565808.96       929957.01
      1564738.36       929789.55      1564210.52       929632.94
#Sta/Elev= 30
  3578.3  896.17  3743.0  883.66  3925.4  858.10  4062.9  849.88  4158.8  839.73
  4204.0  837.40  4314.5  834.10  4402.1  834.50  4411.5  832.80  4430.0  834.96
  4545.1  832.72  4709.1  835.06  4816.0  833.06  4946.3  835.05  4963.1  831.34
  4987.3  830.41  4990.3  825.41  5009.7  825.41  5012.7  830.41  5017.8  833.97
  5047.6  837.34  5081.2  852.63  5097.0  857.44  5107.3  858.12  5183.1  861.88
  5262.0  869.90  5327.1  872.81  5350.7  876.77  5595.9  902.12  5622.1  906.66
#Mann=4,-1,0
  3578.3    0.13       0  4987.3    0.05       0  5012.7    0.13       0
  5107.3    0.07       0
Bank Sta=4987.3,5012.7
XS Rating Curve= 0
Exp/Cntr=0.3,0.1
