HEC-RAS study Grassy Creek.prj: Grassy Creek Limited Detail Study

--- Grassy Creek.g01 (geometry) --- (continued)

Type RM Length L Ch R = 1,19418,829,829,829
BEGIN DESCRIPTION:
Grassy Creek 41.0
END DESCRIPTION:
XS GIS Cut Line= 3
      1565991.34       929157.30      1565834.69       929041.26
      1564581.77       929099.27
#Sta/Elev= 30
  4177.1  906.33  4221.7  902.21  4283.2  893.32  4345.8  889.72  4393.2  884.90
  4429.9  876.87  4512.2  854.66  4544.7  844.37  4564.4  840.15  4607.1  834.93
  4704.8  829.88  4950.5  830.36  4987.0  826.27  4990.0  821.27  5010.0  821.27
  5013.0  826.27  5048.5  829.38  5210.7  832.44  5229.4  833.45  5250.4  839.17
  5343.6  862.96  5432.7  881.79  5467.0  886.62  5491.1  885.76  5515.4  895.30
  5529.2  897.99  5572.2  902.74  5600.7  904.15  5606.1  905.88  5626.3  905.04
#Mann=6,-1,0
  4177.1    0.13       0  4987.0    0.05       0  5013.0    0.13       0
  5048.5    0.07       0  5250.4    0.13       0  5467.0    0.07       0
Bank Sta=4987,5013
XS Rating Curve= 0
Exp/Cntr=0.3,0.1

Type RM Length L Ch R = 1,18589,505,505,505
BEGIN DESCRIPTION:
Grassy Creek 40.0
END DESCRIPTION:
XS GIS Cut Line= 4
      1565596.90       928246.55      1565446.04       928298.77
      1564958.78       928316.18      1564604.98       928287.18
#Sta/Elev= 30
  4642.3  913.05  4720.2  892.85  4743.1  883.08  4794.3  868.47  4876.6  839.91
  4901.9  833.17  4913.3  828.81  4927.3  825.73  4962.8  827.58  4973.2  823.89
  4986.7  822.78  4989.7  817.78  5010.3  817.78  5013.3  822.78  5022.2  824.37
  5030.3  828.13  5044.3  831.15  5067.3  834.01  5094.3  836.50  5152.6  838.62
  5165.6  840.13  5187.6  838.46  5202.0  839.96  5218.7  844.60  5260.0  851.09
  5327.9  863.91  5392.4  877.53  5482.1  892.70  5571.0  900.55  5644.5  902.48
#Mann=4,-1,0
  4642.3    0.13       0  4986.7    0.05       0  5013.3    0.13       0
  5067.3    0.07       0
Bank Sta=4986.7,5013.3
XS Rating Curve= 0
Exp/Cntr=0.3,0.1

Type RM Length L Ch R = 1,18084,605,605,605
BEGIN DESCRIPTION:
Grassy Creek 39.0
END DESCRIPTION:
XS GIS Cut Line= 5
      1565741.70       927913.01      1565287.19       927834.73
      1564905.86       927852.41      1564761.92       927945.84
      1564676.09       928107.41
#Sta/Elev= 30
  4617.0  892.77  4676.5  886.14  4810.1  866.73  4820.5  862.95  4825.5  863.06
  4845.1  859.59  4887.3  850.52  4937.7  832.66  4953.3  828.59  4964.1  827.10
  4986.7  820.84  4989.7  815.84  5010.3  815.84  5013.3  820.84  5034.2  825.97
  5059.0  825.61  5152.6  825.15  5232.8  826.17  5260.4  827.19  5313.0  830.80
  5341.5  835.99  5369.7  835.51  5386.0  839.19  5398.4  840.37  5427.8  842.76
  5472.5  844.33  5524.7  849.12  5565.4  856.36  5660.1  869.61  5814.5  887.42
#Mann=4,-1,0
  4617.0    0.13       0  4986.7    0.05       0  5013.3    0.13       0
  5059.0    0.07       0
Bank Sta=4986.7,5013.3
XS Rating Curve= 0
Exp/Cntr=0.3,0.1

Type RM Length L Ch R = 1,17479,294,294,294
BEGIN DESCRIPTION:
Grassy Creek 38.0
END DESCRIPTION:
XS GIS Cut Line= 5
      1565903.37       927806.96      1565749.32       927572.10
      1565524.57       927382.70      1565375.58       927180.67
      1565340.22       926920.58
#Sta/Elev= 30
  4543.7  894.62  4604.0  885.02  4667.7  878.25  4708.9  867.60  4779.2  852.69
  4861.7  841.85  4882.3  834.19  4891.5  837.66  4914.8  834.99  4941.0  826.78
  4960.4  825.52  4986.7  819.43  4989.7  814.43  5010.3  814.43  5013.3  819.43
  5039.7  821.62  5047.1  823.38  5069.5  824.06  5139.8  821.61  5203.5  822.16
  5229.9  822.51  5235.7  823.70  5247.8  821.62  5324.1  822.86  5339.5  824.61
  5390.1  838.32  5415.1  842.71  5494.0  853.79  5533.2  861.25  5632.0  876.75
#Mann=5,-1,0
  4543.7    0.13       0  4986.7    0.05       0  5013.3    0.13       0
  5203.5    0.07       0  5324.1    0.13       0
Bank Sta=4986.7,5013.3
XS Rating Curve= 0
Exp/Cntr=0.3,0.1

Type RM Length L Ch R = 1,17185,538,538,538
BEGIN DESCRIPTION:
Grassy Creek 37.0
END DESCRIPTION:
XS GIS Cut Line= 4
      1566064.99       927655.43      1565900.84       927438.25
      1565527.09       927016.52      1565373.06       926842.29
#Sta/Elev= 30
  4393.9  886.13  4408.9  886.16  4444.1  879.96  4490.2  876.11  4519.8  875.54
  4554.3  872.03  4614.5  869.27  4671.8  864.18  4717.2  854.71  4755.2  844.71
  4801.4  827.42  4825.4  823.08  4959.7  822.32  4986.3  817.86  4989.3  812.86
  5010.7  812.86  5013.7  817.86  5028.3  822.23  5052.7  819.34  5091.4  820.49
  5117.1  821.75  5171.8  828.17  5189.7  831.00  5269.9  848.09  5284.5  849.38
  5373.7  867.96  5391.1  872.86  5410.9  876.02  5440.9  883.30  5462.2  887.11
#Mann=5,-1,0
  4393.9    0.13       0  4986.3    0.05       0  5013.7    0.13       0
  5028.3    0.07       0  5171.8    0.13       0
Bank Sta=4986.3,5013.7
XS Rating Curve= 0
Exp/Cntr=0.3,0.1

Type RM Length L Ch R = 1,16647,396,396,396
BEGIN DESCRIPTION:
Grassy Creek 36.0
END DESCRIPTION:
XS GIS Cut Line= 3
      1566342.80       927370.11      1566201.36       927072.08
      1565880.24       926468.70
#Sta/Elev= 30
  4418.6  887.97  4536.9  873.77  4633.8  858.24  4642.3  857.75  4686.4  848.69
  4775.4  833.44  4795.9  827.31  4834.2  820.52  4871.2  819.30  4923.9  820.07
  4942.6  817.56  4963.9  817.93  4986.3  816.22  4989.3  811.22  5010.7  811.22
  5013.7  816.22  5026.2  816.13  5045.6  818.46  5078.1  820.66  5119.2  819.62
  5164.8  821.28  5172.1  822.71  5185.0  826.62  5187.4  828.68  5237.2  852.17
  5245.8  853.71  5257.7  858.90  5279.5  865.14  5359.7  886.04  5432.0  897.00
#Mann=5,-1,0
  4418.6    0.13       0  4986.3    0.05       0  5013.7    0.13       0
  5045.6    0.07       0  5119.2    0.13       0
Bank Sta=4986.3,5013.7
XS Rating Curve= 0
Exp/Cntr=0.3,0.1

Type RM Length L Ch R = 1,16251,390,390,390
BEGIN DESCRIPTION:
Grassy Creek 35.0
END DESCRIPTION:
XS GIS Cut Line= 5
      1566428.63       927299.39      1566519.55       926930.66
      1566408.43       926604.90      1566383.18       926577.12
      1566188.75       926567.02
#Sta/Elev= 30
  4413.4  876.77  4512.3  860.86  4611.1  848.88  4636.1  843.74  4732.2  830.94
  4782.3  828.50  4800.7  829.31  4832.5  827.94  4855.2  824.89  4880.3  819.45
  4905.5  817.71  4960.7  817.29  4980.0  815.45  4986.3  814.23  4989.3  809.23
  5010.7  809.23  5013.7  814.23  5032.0  814.88  5038.0  816.18  5062.2  814.69
  5070.8  815.72  5086.1  820.99  5092.6  824.45  5106.5  834.57  5114.7  841.68
  5164.8  854.99  5181.9  857.02  5194.5  856.29  5299.4  863.20  5369.6  874.07
#Mann=5,-1,0
  4413.4    0.13       0  4905.5    0.07       0  4980.0    0.13       0
  4986.3    0.05       0  5013.7    0.13       0
Bank Sta=4986.3,5013.7
XS Rating Curve= 0
Exp/Cntr=0.3,0.1

Type RM Length L Ch R = 1,15861,490,490,490
BEGIN DESCRIPTION:
Grassy Creek 34.0
END DESCRIPTION:
XS GIS Cut Line= 4
      1567080.18       926498.83      1566542.28       926513.98
      1566393.28       926569.54      1566165.96       926556.91
#Sta/Elev= 30
  4667.5  904.18  4715.4  896.85  4755.1  886.87  4764.5  883.32  4792.5  871.80
  4826.5  855.61  4851.8  841.72  4877.8  824.38  4884.2  821.06  4899.8  816.50
  4969.4  815.01  4986.3  811.45  4989.3  806.45  5010.7  806.45  5013.7  811.45
  5029.0  814.13  5067.1  817.24  5097.2  816.61  5167.4  819.17  5207.1  825.24
  5235.2  833.55  5272.8  840.87  5293.5  847.58  5334.3  854.76  5379.2  857.97
  5398.3  856.84  5456.8  859.79  5505.0  864.20  5570.1  875.10  5592.3  876.84
#Mann=5,-1,0
  4667.5    0.13       0  4877.8    0.07       0  4969.4    0.13       0
  4986.3    0.05       0  5013.7    0.13       0
Bank Sta=4986.3,5013.7
XS Rating Curve= 0
Exp/Cntr=0.3,0.1

Type RM Length L Ch R = 1,15371,490,490,490
BEGIN DESCRIPTION:
Grassy Creek 33.0
END DESCRIPTION:
XS GIS Cut Line= 6
      1566408.42       925766.47      1566552.38       925988.72
      1566610.46       926309.43      1566522.07       926486.21
      1566400.86       926556.91      1566161.00       926534.19
#Sta/Elev= 30
  4538.3  851.10  4598.5  847.94  4696.7  845.93  4750.2  838.75  4786.4  832.32
  4874.7  821.06  4913.6  815.66  4973.1  815.08  4979.2  812.91  4986.3  810.39
  4989.3  805.39  5010.7  805.39  5013.7  810.39  5044.2  810.80  5068.6  813.14
  5142.0  812.28  5157.1  816.10  5191.7  818.65  5237.9  819.14  5262.7  820.18
  5330.9  828.85  5372.5  836.98  5398.4  844.67  5450.3  855.14  5480.6  857.68
  5515.3  856.05  5601.4  861.37  5622.8  864.11  5645.6  870.22  5709.0  877.58
#Mann=8,-1,0
  4538.3    0.07       0  4598.5    0.13       0  4874.7    0.07       0
  4979.2    0.13       0  4986.3    0.05       0  5013.7    0.13       0
  5191.7    0.07       0  5237.9    0.13       0
Bank Sta=4986.3,5013.7
XS Rating Curve= 0
Exp/Cntr=0.3,0.1

Type RM Length L Ch R = 1,14881,437,437,437
BEGIN DESCRIPTION:
Grassy Creek 32.0
END DESCRIPTION:
XS GIS Cut Line= 4
      1566274.59       925796.79      1566178.63       926127.61
      1566097.82       926289.23      1565928.60       926412.99
#Sta/Elev= 30
  4517.8  850.99  4560.3  848.24  4573.1  848.14  4592.8  846.04  4633.3  844.93
  4733.1  833.69  4756.8  829.64  4767.4  829.21  4794.6  824.81  4817.8  822.86
  4844.9  821.87  4895.6  816.31  4930.1  815.81  4956.3  813.01  4977.6  810.12
  4986.3  806.85  4989.3  801.85  5010.7  801.85  5013.7  806.85  5038.3  816.19
  5043.0  819.73  5048.9  825.25  5068.3  835.82  5086.9  845.03  5096.5  848.23
  5113.3  855.34  5160.4  870.79  5177.0  874.17  5209.4  884.97  5252.6  894.46
#Mann=5,-1,0
  4517.8    0.07       0  4560.3    0.13       0  4956.3    0.13       0
  4986.3    0.05       0  5013.7    0.13       0
Bank Sta=4986.3,5013.7
XS Rating Curve= 0
Exp/Cntr=0.3,0.1

Type RM Length L Ch R = 1,14444,326,326,326
BEGIN DESCRIPTION:
Grassy Creek 31.0
END DESCRIPTION:
XS GIS Cut Line= 4
      1566274.55       925751.36      1566181.15       925822.04
      1565875.59       925859.92      1565779.61       925973.59
#Sta/Elev= 30
  4700.4  855.65  4748.9  852.17  4771.8  849.04  4779.1  847.60  4794.0  845.11
  4807.1  841.77  4824.0  839.05  4853.8  833.11  4900.8  822.87  4917.5  817.65
  4934.8  814.12  4951.2  809.92  4960.2  810.14  4960.9  809.73  4986.3  806.49
  4989.3  801.49  5010.7  801.49  5013.7  806.49  5033.8  809.60  5054.4  816.01
  5070.2  822.74  5079.7  828.61  5099.2  836.89  5110.8  842.95  5137.9  855.29
  5155.9  862.39  5185.7  872.09  5220.6  879.98  5241.0  883.94  5274.2  889.15
#Mann=5,-1,0
  4700.4    0.07       0  4779.1    0.13       0  4900.8    0.13       0
  4986.3    0.05       0  5013.7    0.13       0
Bank Sta=4986.3,5013.7
XS Rating Curve= 0
Exp/Cntr=0.3,0.1

Type RM Length L Ch R = 1,14118,217,217,217
BEGIN DESCRIPTION:
Grassy Creek 30.0
END DESCRIPTION:
XS GIS Cut Line= 3
      1566267.00       925493.75      1565814.98       925536.68
      1565597.79       925630.13
#Sta/Elev= 30
  4679.0  877.69  4736.8  868.73  4753.0  863.98  4771.1  856.71  4784.9  854.25
  4805.3  853.70  4817.2  852.08  4837.1  845.55  4940.5  815.80  4959.3  810.73
  4968.0  809.40  4981.0  809.42  4985.5  807.58  4986.3  804.43  4989.3  799.43
  5010.7  799.43  5013.7  804.43  5033.1  804.90  5039.3  807.18  5060.7  811.00
  5080.5  816.06  5101.3  822.84  5122.0  827.03  5176.9  835.05  5211.2  836.61
  5223.8  838.80  5236.4  843.30  5295.3  857.11  5343.3  864.08  5369.5  866.78
#Mann=6,-1,0
  4679.0    0.07       0  4817.2    0.13       0  4940.5    0.13       0
  4986.3    0.05       0  5013.7    0.13       0  5223.8    0.13       0
Bank Sta=4986.3,5013.7
XS Rating Curve= 0
Exp/Cntr=0.5,0.3

Type RM Length L Ch R = 1,13901,80,80,80
BEGIN DESCRIPTION:
Grassy Creek Rd (GC) us
END DESCRIPTION:
XS GIS Cut Line= 5
      1566246.43       925472.94      1566098.14       925416.77
      1566041.96       925349.36      1565498.16       925252.73
      1565215.06       925358.33
#Sta/Elev= 30
  4592.6  876.37  4622.6  872.17  4667.3  863.42  4692.8  853.89  4713.9  847.23
  4736.8  844.91  4747.4  842.57  4761.3  841.54  4825.1  830.66  4838.9  829.65
  4870.2  820.88  4887.9  815.89  4916.8  810.44  4949.4  808.67  4980.0  804.90
  4990.0  798.20  5010.0  798.20  5020.0  804.90  5020.7  806.97  5040.3  809.05
  5084.2  816.80  5134.6  818.79  5157.7  818.12  5261.6  821.03  5292.3  823.19
  5374.2  826.39  5403.8  828.84  5487.2  831.48  5602.1  836.85  5693.4  840.93
#Mann=6,-1,0
  4592.6    0.07       0  4870.2    0.13       0  4980.0    0.05       0
  5020.0    0.13       0  5261.6    0.07       0  5602.1    0.13       0
#XS Ineff=2,0
    0.00 4939.00  820.58 5061.00    0.00  817.30
Permanent Ineff=
       F       F
Bank Sta=4980,5020
XS Rating Curve= 0
Exp/Cntr=0.5,0.3

Type RM Length L Ch R =3,13855,,,
BEGIN DESCRIPTION:
Grassy Creek Rd (GC) TOR
Structure ID: LDS_GC_03
Approximate Survey Structure
END DESCRIPTION:
Bridge Culvert--1,0,-1,-1,0
Deck Dist Width WeirC Skew NumUp NumDn MinLoCord MaxHiCord MaxSubmerge Is_Ogee
36,20,3,,16,16,,,0.95,0,1,1,,,
  4563.6  4649.1  4709.3  4726.0  4890.2  4941.9  4965.4  4975.0  4975.0  5025.0
  5025.0  5149.7  5244.6  5395.9  5560.8  5743.8
  878.40  864.56  845.96  843.46  824.68  820.28  817.30  817.30  817.30  817.30
  817.30  817.30  819.81  825.94  833.39  842.25
  778.20  778.20  778.20  778.20  778.20  778.20  778.20  778.20  815.30  815.30
  778.20  778.20  778.20  778.20  778.20  778.20
  4563.6  4649.1  4709.3  4726.0  4890.2  4941.9  4965.4  4975.0  4975.0  5025.0
  5025.0  5149.7  5244.6  5395.9  5560.8  5743.8
  878.40  864.56  845.96  843.46  824.68  820.28  817.30  817.30  817.30  817.30
  817.30  817.30  819.81  825.94  833.39  842.25
  778.20  778.20  778.20  778.20  778.20  778.20  778.20  778.20  815.30  815.30
  778.20  778.20  778.20  778.20  778.20  778.20
BR Coef=1,1,0,1.25,0,,,0.8,0,2,0,
WSPro=,,,, 1 ,,,, 0 ,,,, 0 ,,,,-1 ,-1 ,-1 , 0 , 0 , 0 , 0 , 0
BC Design=,,0,,0,,,,,,

Type RM Length L Ch R = 1,13821,140,140,140
BEGIN DESCRIPTION:
Grassy Creek Rd (GC) ds
END DESCRIPTION:
XS GIS Cut Line= 6
      1566248.68       925441.48      1566131.84       925374.07
      1566084.65       925279.70      1565817.25       925228.01
      1565484.68       925196.55      1565197.06       925335.87
#Sta/Elev= 30
  4558.7  878.55  4592.9  873.61  4657.5  860.42  4693.6  849.57  4717.2  847.37
  4727.2  848.44  4772.9  838.00  4844.8  828.79  4868.8  821.02  4921.6  813.85
  4953.3  811.99  4966.2  810.41  4980.0  804.65  4990.0  797.95  5010.0  797.95
  5020.0  804.65  5035.0  808.11  5083.3  810.44  5095.3  812.90  5126.5  814.73
  5159.0  813.35  5184.0  815.40  5225.6  814.69  5280.3  821.34  5392.4  824.29
  5404.2  826.24  5435.8  825.85  5658.2  837.44  5718.6  840.68  5725.1  841.13
#Mann=7,-1,0
  4558.7    0.07       0  4953.3    0.13       0  4980.0    0.05       0
  5020.0    0.13       0  5280.3    0.07       0  5658.2    0.13       0
  5718.6    0.07       0
#XS Ineff=2,0
    0.00 4951.00  819.79 5049.00    0.00  817.30
Permanent Ineff=
       F       F
Bank Sta=4980,5020
XS Rating Curve= 0
Exp/Cntr=0.5,0.3

Type RM Length L Ch R = 1,13681,300,300,300
BEGIN DESCRIPTION:
Grassy Creek 29.0
END DESCRIPTION:
XS GIS Cut Line= 4
      1566309.97       925114.95      1566072.57       925097.28
      1565580.13       925114.95      1565181.13       925327.08
#Sta/Elev= 30
  4549.5  875.73  4634.3  858.48  4646.9  857.25  4695.6  844.58  4707.6  842.51
  4720.7  838.74  4774.4  826.27  4849.2  815.14  4885.1  813.08  4917.2  809.79
  4954.7  809.54  4966.0  809.55  4986.1  806.27  4986.3  802.72  4989.3  797.72
  5010.7  797.72  5013.7  802.72  5055.2  808.16  5082.0  807.09  5210.6  807.28
  5236.6  808.95  5274.3  816.88  5287.7  819.43  5314.7  821.95  5416.8  824.73
  5437.2  826.00  5452.5  824.56  5466.9  828.65  5538.7  830.62  5732.2  840.69
#Mann=7,-1,0
  4549.5    0.07       0  4954.7    0.13       0  4986.3    0.05       0
  5013.7    0.13       0  5082.0    0.07       0  5210.6    0.13       0
  5274.3    0.07       0
#XS Ineff=2,0
       0                 5053.10    0.00  821.88
Permanent Ineff=
       F       F
Bank Sta=4986.3,5013.7
XS Rating Curve= 0
Exp/Cntr=0.3,0.1

Type RM Length L Ch R = 1,13381,808,808,808
BEGIN DESCRIPTION:
Grassy Creek 28.0
END DESCRIPTION:
XS GIS Cut Line= 5
      1566327.62       924847.27      1566053.50       924789.40
      1565510.08       924875.70      1565270.34       924971.60
      1564963.44       925208.17
#Sta/Elev= 30
  4418.3  888.94  4484.4  880.99  4516.7  872.69  4556.2  864.68  4579.8  858.06
  4649.1  835.58  4695.7  816.66  4728.7  808.66  4802.9  805.83  4862.5  806.07
  4910.2  808.22  4962.8  807.57  4975.8  805.69  4986.2  802.11  4989.2  797.11
  5010.8  797.11  5013.8  802.11  5037.2  806.90  5059.9  806.00  5155.3  805.91
  5215.8  812.35  5499.4  818.19  5518.8  820.44  5576.8  832.05  5609.7  834.73
  5646.6  842.30  5739.9  847.95  5844.7  851.59  5857.3  853.91  5894.4  856.30
#Mann=6,-1,0
  4418.3    0.13       0  4516.7    0.07       0  4962.8    0.13       0
  4986.2    0.05       0  5013.8    0.13       0  5059.9    0.07       0
#XS Ineff=2,0
    0.00 4830.10  823.62               0
Permanent Ineff=
       F       F
Bank Sta=4986.2,5013.8
XS Rating Curve= 0
Exp/Cntr=0.3,0.1

Type RM Length L Ch R = 1,12573,475,475,475
BEGIN DESCRIPTION:
Grassy Creek 27.0
END DESCRIPTION:
XS GIS Cut Line= 3
      1566072.56       924195.73      1565706.39       924324.53
      1565659.23       924362.64
#Sta/Elev= 30
  4692.8  866.00  4703.7  864.97  4715.2  864.59  4726.8  863.41  4738.5  861.42
  4768.1  859.53  4807.5  854.86  4827.4  851.88  4839.6  849.43  4860.8  843.98
  4872.6  841.58  4888.2  836.77  4923.5  817.48  4941.0  809.17  4954.5  804.77
  4959.7  802.46  4986.2  799.40  4989.2  794.40  5010.8  794.40  5013.8  799.40
  5014.9  801.22  5016.6  801.72  5030.2  802.74  5044.2  802.22  5050.6  802.70
  5057.5  803.58  5069.7  807.60  5092.4  810.55  5126.0  816.15  5141.6  816.33
#Mann=3,-1,0
  4692.8    0.13       0  4986.2    0.05       0  5013.8    0.13       0
Bank Sta=4986.2,5013.8
XS Rating Curve= 0
Exp/Cntr=0.3,0.1

Type RM Length L Ch R = 1,12098,397,397,397
BEGIN DESCRIPTION:
Grassy Creek 26.0
END DESCRIPTION:
XS GIS Cut Line= 4
      1566019.58       924167.98      1565817.51       924056.84
      1565633.16       923880.07      1565618.01       923680.57
#Sta/Elev= 30
  4597.6  861.52  4627.8  856.43  4663.3  849.30  4669.4  847.22  4684.4  844.46
  4705.0  839.09  4709.4  838.83  4750.3  829.51  4766.1  824.54  4770.8  824.33
  4792.6  818.40  4829.8  811.47  4889.0  803.99  4910.1  802.97  4949.9  799.52
  4969.7  799.74  4985.3  796.65  4990.2  791.65  5009.8  791.65  5014.7  796.65
  5039.9  804.15  5063.8  809.78  5083.6  819.82  5106.8  829.11  5131.3  838.03
  5194.1  858.08  5202.2  860.40  5221.6  863.91  5272.3  877.62  5283.7  879.82
#Mann=4,-1,0
  4597.6    0.13       0  4985.3    0.05       0  5014.7    0.13       0
  5194.1    0.07       0
Bank Sta=4985.3,5014.7
XS Rating Curve= 0
Exp/Cntr=0.3,0.1

Type RM Length L Ch R = 1,11701,495,495,495
BEGIN DESCRIPTION:
Grassy Creek 25.0
END DESCRIPTION:
XS GIS Cut Line= 4
      1566244.29       923965.93      1566102.87       923791.68
      1565905.89       923632.59      1565761.94       923561.87
#Sta/Elev= 30
  4644.9  872.79  4660.9  871.04  4671.2  868.55  4679.5  867.18  4715.9  858.79
  4720.8  858.01  4727.2  856.16  4760.3  849.69  4795.2  841.56  4803.7  840.06
  4835.8  831.64  4841.0  830.55  4861.5  824.04  4900.0  813.96  4920.4  807.31
  4931.4  804.41  4985.6  793.61  4988.6  788.61  5011.4  788.61  5014.4  793.61
  5020.3  798.85  5060.3  802.39  5082.9  809.29  5118.4  821.51  5153.6  835.20
  5175.3  843.03  5200.0  850.90  5218.1  857.45  5257.8  870.03  5282.9  876.83
#Mann=3,-1,0
  4644.9    0.13       0  4985.6    0.05       0  5014.4    0.13       0
Bank Sta=4985.6,5014.4
XS Rating Curve= 0
Exp/Cntr=0.3,0.1

Type RM Length L Ch R = 1,11206,378,378,378
BEGIN DESCRIPTION:
Grassy Creek 24.0
END DESCRIPTION:
XS GIS Cut Line= 4
      1566517.02       923935.63      1566562.48       923622.48
      1566241.76       923248.74      1566196.30       923064.37
#Sta/Elev= 30
  4328.9  871.91  4348.4  870.73  4440.8  857.31  4480.3  850.71  4645.3  819.03
  4672.8  816.37  4713.5  810.21  4756.3  805.78  4812.9  804.14  4895.3  798.48
  4901.1  799.16  4916.2  797.79  4940.9  797.21  4954.8  797.94  4980.2  796.94
  4985.6  793.01  4988.6  788.01  5011.4  788.01  5014.4  793.01  5038.6  797.30
  5057.6  805.31  5064.0  809.60  5072.3  812.97  5106.9  822.93  5116.6  826.69
  5139.6  833.02  5184.7  840.72  5231.2  851.51  5303.4  866.45  5327.7  870.75
#Mann=4,-1,0
  4328.9    0.13       0  4985.6    0.05       0  5014.4    0.13       0
  5139.6    0.07       0
Bank Sta=4985.6,5014.4
XS Rating Curve= 0
Exp/Cntr=0.3,0.1

Type RM Length L Ch R = 1,10828,473,473,473
BEGIN DESCRIPTION:
Grassy Creek 23.0
END DESCRIPTION:
XS GIS Cut Line= 3
      1566829.26       923625.91      1566667.15       923171.99
      1566398.35       922837.13
#Sta/Elev= 30
  4467.6  833.08  4547.1  822.47  4607.0  808.24  4647.5  802.80  4686.3  798.94
  4764.5  796.30  4771.4  796.61  4822.7  795.37  4886.0  795.07  4905.8  795.90
  4966.6  796.59  4985.6  790.38  4988.6  785.38  5011.4  785.38  5014.4  790.38
  5043.9  797.54  5048.2  799.80  5052.5  801.90  5068.2  802.27  5085.9  803.59
  5151.2  813.80  5164.4  817.05  5176.1  820.94  5185.5  824.09  5223.3  834.38
  5239.4  836.54  5261.1  840.91  5268.1  842.93  5344.4  860.11  5379.0  865.50
#Mann=5,-1,0
  4467.6    0.13       0  4985.6    0.05       0  5014.4    0.13       0
  5048.2    0.07       0  5176.1    0.13       0
#XS Ineff=2,0
    0.00 4820.30  817.27               0
Permanent Ineff=
       F       F
Bank Sta=4985.6,5014.4
XS Rating Curve= 0
Exp/Cntr=0.3,0.1

Type RM Length L Ch R = 1,10355,434,434,434
BEGIN DESCRIPTION:
Grassy Creek 22.0
END DESCRIPTION:
XS GIS Cut Line= 5
      1567284.72       923188.12      1567186.23       923011.36
      1566878.14       922794.18      1566746.83       922733.57
      1566567.52       922675.48
#Sta/Elev= 30
  4610.3  865.34  4624.2  864.19  4678.6  855.90  4700.4  851.75  4733.9  842.70
  4757.0  834.89  4817.8  806.41  4826.0  803.33  4845.5  798.15  4865.1  794.50
  4885.4  792.02  4897.5  791.60  4925.0  794.05  4966.3  793.57  4970.1  791.79
  4985.1  788.59  4988.1  783.59  5011.9  783.59  5014.9  788.59  5032.8  792.41
  5038.4  794.36  5108.5  795.76  5209.3  801.02  5270.5  805.19  5287.8  807.60
  5379.5  823.34  5401.3  828.67  5432.2  831.55  5480.4  841.56  5522.7  847.08
#Mann=5,-1,0
  4610.3    0.13       0  4985.1    0.05       0  5014.9    0.13       0
  5032.8    0.07       0  5287.8    0.13       0
Bank Sta=4985.1,5014.9
XS Rating Curve= 0
Exp/Cntr=0.3,0.1

Type RM Length L Ch R = 1,9921,254,254,254
BEGIN DESCRIPTION:
Grassy Creek 21.0
END DESCRIPTION:
XS GIS Cut Line= 4
      1567418.57       922771.45      1567299.87       922642.66
      1567047.34       922529.02      1566880.65       922425.47
#Sta/Elev= 30
  4707.3  850.81  4712.3  849.95  4732.0  844.57  4737.6  844.05  4787.4  835.64
  4804.7  831.61  4816.1  830.05  4838.0  825.81  4845.4  823.30  4871.9  817.41
  4885.0  813.60  4906.0  808.48  4918.1  804.32  4927.4  802.48  4939.6  798.26
  4958.6  790.74  4985.1  786.51  4988.1  781.51  5011.9  781.51  5014.9  786.51
  5026.3  788.08  5038.0  792.98  5068.7  797.17  5089.0  801.63  5103.5  803.43
  5112.3  803.52  5124.1  804.94  5195.4  814.60  5318.1  845.98  5355.6  851.84
#Mann=3,-1,0
  4707.3    0.13       0  4985.1    0.05       0  5014.9    0.13       0
Bank Sta=4985.1,5014.9
XS Rating Curve= 0
Exp/Cntr=0.3,0.1

Type RM Length L Ch R = 1,9667,511,511,511
BEGIN DESCRIPTION:
Grassy Creek 20.0
END DESCRIPTION:
XS GIS Cut Line= 5
      1567575.15       922753.80      1567438.77       922508.81
      1567304.93       922357.30      1566989.26       922407.80
      1566890.73       922405.28
#Sta/Elev= 30
  4604.3  846.48  4636.2  843.28  4664.1  839.50  4708.2  835.20  4724.2  832.38
  4789.0  824.21  4875.7  807.07  4908.9  799.26  4939.8  794.42  4969.3  791.91
  4985.1  784.30  4988.1  779.30  5011.9  779.30  5014.9  784.30  5033.7  785.50
  5037.1  787.54  5048.7  796.91  5053.7  800.12  5139.8  807.68  5148.9  807.24
  5161.1  808.67  5170.1  808.22  5220.5  815.52  5383.5  830.10  5407.4  831.54
  5423.0  836.16  5449.6  840.70  5472.6  842.60  5494.7  847.34  5505.1  848.50
#Mann=6,-1,0
  4604.3    0.13       0  4636.2    0.15       0  4939.8    0.13       0
  4985.1    0.05       0  5014.9    0.13       0  5037.1    0.07       0
Bank Sta=4985.1,5014.9
XS Rating Curve= 0
Exp/Cntr=0.3,0.1

Type RM Length L Ch R = 1,9156,269,269,269
BEGIN DESCRIPTION:
Grassy Creek 19.0
END DESCRIPTION:
XS GIS Cut Line= 5
      1567587.74       921922.98      1567476.65       922223.45
      1567268.65       922354.21      1567067.31       922391.96
      1566968.48       922402.74
#Sta/Elev= 30
  4801.6  865.46  4814.8  864.47  4827.1  860.17  4864.5  841.55  4897.2  830.06
  4918.1  820.99  4923.1  819.52  4939.7  810.04  4954.4  797.72  4958.1  794.08
  4965.7  788.29  4975.1  783.20  4984.3  782.61  4987.3  777.61  5012.7  777.61
  5015.7  782.61  5033.0  784.72  5055.1  789.87  5067.6  790.21  5144.7  794.95
  5168.3  795.81  5173.1  796.97  5280.1  799.67  5334.7  802.16  5355.3  805.13
  5374.1  806.53  5393.2  806.01  5457.7  814.41  5649.2  832.09  5671.9  836.51
#Mann=5,-1,0
  4801.6    0.07       0  4827.1    0.13       0  4984.3    0.05       0
  5015.7    0.13       0  5067.6    0.07       0
Bank Sta=4984.3,5015.7
XS Rating Curve= 0
Exp/Cntr=0.5,0.3

Type RM Length L Ch R = 1,8887,57,57,57
BEGIN DESCRIPTION:
Hauser Rd (GC) us
END DESCRIPTION:
XS GIS Cut Line= 6
      1567265.04       921645.96      1567239.88       921737.60
      1567250.67       922293.08      1567207.53       922345.22
      1567135.62       922375.78      1567002.56       922397.35
#Sta/Elev= 30
  4565.7  836.65  4583.4  836.17  4617.0  832.34  4657.4  823.08  4676.5  820.81
  4684.3  818.59  4699.2  818.35  4713.4  814.57  4726.2  812.93  4734.3  814.00
  4752.2  812.46  4778.3  806.52  4812.5  804.05  4851.9  796.37  4875.7  794.95
  4896.1  795.77  4924.5  789.24  4950.2  786.55  4957.6  783.89  4980.0  782.70
  4989.0  777.70  5003.5  777.70  5011.5  782.70  5012.6  786.04  5059.7  793.32
  5084.1  793.70  5090.4  795.21  5103.2  794.94  5205.4  801.48  5497.4  831.42
#Mann=3,-1,0
  4565.7    0.13       0  4980.0    0.05       0  5011.5    0.07       0
#XS Ineff=2,0
    0.00 4922.00  794.50 5078.00    0.00  794.50
Permanent Ineff=
       F       F
Bank Sta=4980,5011.5
XS Rating Curve= 0
Exp/Cntr=0.5,0.3

Type RM Length L Ch R =3,8860,,,
BEGIN DESCRIPTION:
Hauser Rd (GC) TOR
Structure ID: LDS_GC_02
Approximate Survey Structure
END DESCRIPTION:
Bridge Culvert--1,0,-1,-1,0
Deck Dist Width WeirC Skew NumUp NumDn MinLoCord MaxHiCord MaxSubmerge Is_Ogee
13,28,3,,16,16,,,0.95,0,1,1,,,
  4511.5  4579.8  4657.6  4731.4  4831.2  4867.4  4935.0  4935.0  5065.0  5065.0
  5088.3  5160.9  5235.4  5333.2  5408.6  5496.2
  828.43  821.74  813.76  804.99  796.51  794.50  794.50  794.50  794.50  794.50
  794.50  798.38  803.78  816.17  823.87  833.51
  757.70  757.70  757.70  757.70  757.70  757.70  757.70  792.50  792.50  757.70
  757.70  757.70  757.70  757.70  757.70  757.70
  4511.5  4579.8  4657.6  4731.4  4831.2  4867.4  4935.0  4935.0  5065.0  5065.0
  5088.3  5160.9  5235.4  5333.2  5408.6  5496.2
  828.43  821.74  813.76  804.99  796.51  794.50  794.50  794.50  794.50  794.50
  794.50  798.38  803.78  816.17  823.87  833.51
  757.70  757.70  757.70  757.70  757.70  757.70  757.70  792.50  792.50  757.70
  757.70  757.70  757.70  757.70  757.70  757.70
Pier Skew, UpSta & Num, DnSta & Num=,4967.5,2,4967.5,2,0,0,0,0,0
       1       1
  780.71  792.50
       1       1
  784.23  792.50
Pier Skew, UpSta & Num, DnSta & Num=,5032.5,2,5032.5,2,0,0,0,0,0
       1       1
  787.56  792.50
       1       1
  785.48  792.50
Abutment Skew #Up #Dn=,2,2
  4935.0  4952.5
  792.50  785.72
  4935.0  4952.5
  792.50  783.76
Abutment Skew #Up #Dn=,2,2
  5047.5  5065.0
  791.34  792.50
  5047.5  5065.0
  793.23  792.50
BR Coef=1,1,0,1.25,0,,,0.8,0,2,0,
WSPro=,,,, 1 ,,,, 0 ,,,, 0 ,,,,-1 ,-1 ,-1 , 0 , 0 , 0 , 0 , 0
BC Design=,,0,,0,,,,,,

Type RM Length L Ch R = 1,8830,397,397,397
BEGIN DESCRIPTION:
Hauser Rd (GC) ds
END DESCRIPTION:
XS GIS Cut Line= 6
      1567223.69       921608.20      1567173.37       921692.66
      1567203.93       922127.70      1567202.13       922269.71
      1567139.21       922338.03      1567006.19       922375.78
#Sta/Elev= 30
  4531.8  826.44  4606.0  820.21  4623.7  817.50  4632.9  813.96  4691.4  805.35
  4728.6  801.65  4744.0  802.08  4750.5  798.65  4794.6  797.96  4848.5  790.78
  4855.6  791.89  4875.7  789.11  4928.6  788.75  4935.5  787.36  4964.9  783.82
  4980.0  782.45  4989.0  777.45  5003.5  777.45  5011.5  782.45  5043.6  793.62
  5068.5  793.20  5161.5  796.89  5238.2  801.43  5246.7  802.26  5301.1  815.71
  5331.4  820.41  5342.9  819.82  5354.3  822.21  5386.3  824.39  5439.4  830.88
#Mann=5,-1,0
  4531.8    0.13       0  4935.5    0.07       0  4964.9    0.14       0
  4980.0    0.05       0  5011.5    0.07       0
#XS Ineff=2,0
    0.00 4919.00  794.50 5081.00    0.00  794.50
Permanent Ineff=
       F       F
Bank Sta=4980,5011.5
XS Rating Curve= 0
Exp/Cntr=0.5,0.3

Type RM Length L Ch R = 1,8433,498,498,498
BEGIN DESCRIPTION:
Grassy Creek 18.0
END DESCRIPTION:
XS GIS Cut Line= 4
      1567176.11       921415.38      1566953.90       921736.06
      1566756.93       922029.00      1566683.69       922238.63
#Sta/Elev= 30
  4412.5  854.21  4451.2  848.90  4479.9  848.23  4495.6  846.21  4557.7  834.10
  4564.8  831.08  4591.5  826.92  4634.3  823.96  4690.5  815.83  4734.3  813.28
  4792.4  797.58  4803.1  794.31  4850.1  789.26  4906.6  785.65  4957.9  784.64
  4966.4  782.36  4975.2  779.99  4984.3  779.58  4987.3  774.58  5012.7  774.58
  5015.7  779.58  5019.6  784.71  5063.0  787.44  5095.7  793.24  5146.2  805.99
  5189.6  814.26  5236.9  831.14  5269.8  840.15  5318.4  852.00  5377.7  862.36
#Mann=5,-1,0
  4412.5    0.13       0  4792.4    0.07       0  4966.4    0.14       0
  4984.3    0.05       0  5015.7    0.14       0
Bank Sta=4984.3,5015.7
XS Rating Curve= 0
Exp/Cntr=0.3,0.1

Type RM Length L Ch R = 1,7935,417,417,417
BEGIN DESCRIPTION:
Grassy Creek 17.0
END DESCRIPTION:
XS GIS Cut Line= 4
      1566936.25       921228.46      1566587.73       921417.87
      1566340.25       921746.17      1566340.25       921970.88
#Sta/Elev= 30
  4323.5  846.73  4377.3  843.57  4389.6  841.35  4503.0  828.49  4565.0  822.44
  4578.0  819.67  4613.6  815.09  4637.7  813.40  4657.5  808.47  4696.4  802.27
  4746.6  787.89  4773.5  785.34  4828.6  783.47  4882.4  783.27  4913.2  784.28
  4959.6  783.61  4984.3  777.48  4987.3  772.48  5012.7  772.48  5015.7  777.48
  5030.4  779.73  5041.1  783.14  5112.0  808.62  5143.3  818.23  5157.5  821.05
  5183.0  828.90  5208.7  834.74  5260.3  841.45  5317.6  847.42  5356.0  853.40
#Mann=5,-1,0
  4323.5    0.13       0  4746.6    0.07       0  4913.2    0.14       0
  4984.3    0.05       0  5015.7    0.14       0
Bank Sta=4984.3,5015.7
XS Rating Curve= 0
Exp/Cntr=0.3,0.1

Type RM Length L Ch R = 1,7518,461,461,461
BEGIN DESCRIPTION:
Grassy Creek 16.5
END DESCRIPTION:
XS GIS Cut Line= 3
      1566457.88       921135.50      1566012.87       921465.57
      1565956.88       921757.30
#Sta/Elev= 30
  4528.9  815.76  4552.8  810.96  4574.0  809.57  4601.6  804.53  4668.9  796.49
  4717.3  785.81  4733.5  783.76  4783.8  781.86  4843.4  782.14  4867.7  782.46
  4880.9  777.55  4897.6  774.66  4912.9  780.78  4921.0  781.17  4962.2  782.04
  4984.3  777.14  4987.3  772.14  5012.7  772.14  5015.7  777.14  5033.3  781.61
  5055.1  782.32  5085.2  782.25  5134.9  784.44  5178.3  790.29  5196.7  794.43
  5211.1  796.09  5306.5  816.58  5361.8  826.58  5367.8  828.81  5380.0  830.72
#Mann=7,-1,0
  4528.9    0.13       0  4783.8    0.07       0  4843.4    0.14       0
  4984.3    0.05       0  5015.7    0.14       0  5055.1    0.07       0
  5196.7    0.14       0
#XS Ineff=2,0
    0.00 4795.10  794.39               0
Permanent Ineff=
       F       F
Bank Sta=4984.3,5015.7
XS Rating Curve= 0
Exp/Cntr=0.3,0.1

Type RM Length L Ch R = 1,7057,266,266,266
BEGIN DESCRIPTION:
Grassy Creek 16.0
END DESCRIPTION:
XS GIS Cut Line= 4
      1566089.49       920979.29      1565903.83       921064.75
      1565788.89       921035.28      1565612.10       920976.35
#Sta/Elev= 30
  4716.3  816.17  4742.0  814.04  4795.8  806.29  4820.9  800.39  4836.8  797.07
  4847.2  794.24  4874.0  786.08  4887.9  779.99  4923.0  780.74  4932.3  780.17
  4949.8  778.28  4955.9  778.36  4975.0  774.84  4984.3  774.46  4987.3  769.46
  5012.7  769.46  5015.7  774.46  5025.9  776.09  5036.2  780.77  5038.5  782.16
  5048.9  785.93  5059.6  787.04  5066.0  788.10  5080.0  789.04  5083.1  790.96
  5096.2  796.55  5123.4  809.74  5151.3  822.63  5190.5  838.70  5225.7  853.97
#Mann=3,-1,0
  4716.3    0.13       0  4984.3    0.05       0  5015.7    0.13       0
Bank Sta=4984.3,5015.7
XS Rating Curve= 0
Exp/Cntr=0.3,0.1

Type RM Length L Ch R = 1,6791,403,403,403
BEGIN DESCRIPTION:
Grassy Creek 15.0
END DESCRIPTION:
XS GIS Cut Line= 2
      1566327.60       920980.98      1565726.61       920713.31
#Sta/Elev= 30
  4606.5  841.50  4626.2  839.92  4634.8  838.48  4657.1  836.48  4728.5  825.08
  4747.7  821.15  4856.4  804.67  4884.9  799.12  4906.0  794.33  4924.1  789.52
  4958.1  778.69  4984.3  772.71  4987.3  767.71  5012.7  767.71  5015.7  772.71
  5033.8  775.84  5041.2  777.99  5059.8  787.48  5086.7  802.97  5091.7  804.79
  5095.9  807.25  5125.5  820.49  5145.7  828.13  5154.3  833.35  5164.5  835.72
  5184.2  842.34  5195.1  844.98  5213.6  850.86  5249.4  860.24  5264.4  863.56
#Mann=3,-1,0
  4606.5    0.13       0  4984.3    0.05       0  5015.7    0.13       0
Bank Sta=4984.3,5015.7
XS Rating Curve= 0
Exp/Cntr=0.3,0.1

Type RM Length L Ch R = 1,6388,329,329,329
BEGIN DESCRIPTION:
Grassy Creek 14.0
END DESCRIPTION:
XS GIS Cut Line= 3
      1566469.06       920713.32      1566115.50       920435.52
      1565956.42       920415.32
#Sta/Elev= 30
  4666.3  835.40  4719.6  826.66  4750.4  820.18  4771.1  815.30  4789.1  810.46
  4803.7  807.86  4812.3  805.64  4833.0  801.57  4844.3  799.93  4858.2  795.97
  4894.0  786.96  4910.0  782.17  4927.9  779.30  4953.9  773.81  4962.5  772.75
  4984.3  772.00  4987.3  767.00  5012.7  767.00  5015.7  772.00  5038.2  778.86
  5068.3  799.19  5092.5  808.39  5100.7  811.08  5117.3  814.55  5156.3  824.20
  5173.4  827.41  5187.3  829.29  5206.3  833.50  5258.3  839.97  5276.3  841.07
#Mann=3,-1,0
  4666.3    0.13       0  4984.3    0.05       0  5015.7    0.13       0
Bank Sta=4984.3,5015.7
XS Rating Curve= 0
Exp/Cntr=0.3,0.1

Type RM Length L Ch R = 1,6059,487,487,487
BEGIN DESCRIPTION:
Grassy Creek 13.0
END DESCRIPTION:
XS GIS Cut Line= 5
      1566620.54       920412.77      1566529.65       920306.73
      1566484.19       920291.58      1566229.14       920309.26
      1565961.42       920402.70
#Sta/Elev= 30
  4779.8  828.05  4790.3  826.11  4811.1  824.49  4824.4  821.03  4850.0  816.91
  4873.7  812.09  4925.2  803.87  4942.1  796.94  4952.8  790.02  4965.5  782.85
  4973.9  771.59  4984.3  769.72  4987.3  764.72  5012.7  764.72  5015.7  769.72
  5038.6  774.46  5079.5  774.88  5092.7  778.97  5132.1  786.34  5150.0  787.44
  5191.7  788.73  5205.2  790.23  5225.3  791.15  5254.8  795.92  5313.3  811.40
  5355.0  821.50  5386.1  828.02  5431.4  834.31  5468.2  838.30  5506.6  840.67
#Mann=5,-1,0
  4779.8    0.13       0  4984.3    0.05       0  5015.7    0.13       0
  5150.0    0.07       0  5225.3    0.13       0
Bank Sta=4984.3,5015.7
XS Rating Curve= 0
Exp/Cntr=0.3,0.1

Type RM Length L Ch R = 1,5572,555,555,555
BEGIN DESCRIPTION:
Grassy Creek 12.0
END DESCRIPTION:
XS GIS Cut Line= 5
      1566812.47       919847.12      1566643.29       919816.82
      1566322.57       919826.92      1566208.93       920152.68
      1565996.80       920374.92
#Sta/Elev= 30
  4609.5  799.12  4639.1  792.82  4665.7  789.46  4687.0  785.42  4705.6  785.67
  4755.0  781.41  4784.0  780.16  4801.5  778.40  4824.8  773.56  4870.8  771.25
  4888.0  772.16  4951.2  771.57  4984.3  768.75  4987.3  763.75  5012.7  763.75
  5015.7  768.75  5037.7  771.76  5102.3  776.35  5149.4  777.88  5202.3  781.67
  5302.8  785.92  5472.6  786.15  5524.4  787.76  5545.8  789.73  5572.4  795.00
  5606.6  804.44  5643.4  816.71  5677.2  826.32  5695.8  830.56  5754.5  837.33
#Mann=5,-1,0
  4609.5    0.13       0  4984.3    0.05       0  5015.7    0.13       0
  5037.7    0.07       0  5545.8    0.13       0
Bank Sta=4984.3,5015.7
XS Rating Curve= 0
Exp/Cntr=0.3,0.1

Type RM Length L Ch R = 1,5017,451,451,451
BEGIN DESCRIPTION:
Grassy Creek 11.0
END DESCRIPTION:
XS GIS Cut Line= 4
      1566267.01       919354.63      1566330.15       919725.90
      1566198.83       920145.11      1565991.79       920359.73
#Sta/Elev= 30
  4825.1  806.67  4836.9  804.74  4879.3  794.68  4935.6  778.47  4949.9  772.87
  4961.8  770.16  4968.6  767.02  4984.3  764.87  4987.3  759.87  5012.7  759.87
  5015.7  764.87  5037.1  769.10  5082.6  772.08  5114.5  773.41  5151.3  773.67
  5245.3  772.54  5279.9  773.29  5295.9  774.23  5308.2  777.40  5359.1  779.01
  5394.7  782.11  5430.0  783.85  5496.5  785.87  5637.3  785.47  5711.1  787.16
  5728.4  788.03  5741.2  790.04  5762.7  793.58  5881.7  828.79  5939.2  836.12
#Mann=5,-1,0
  4825.1    0.13       0  4984.3    0.05       0  5015.7    0.13       0
  5082.6    0.07       0  5741.2    0.13       0
Bank Sta=4984.3,5015.7
XS Rating Curve= 0
Exp/Cntr=0.3,0.1

Type RM Length L Ch R = 1,4566,485,485,485
BEGIN DESCRIPTION:
Grassy Creek 10.0
END DESCRIPTION:
XS GIS Cut Line= 3
      1566193.76       919342.08      1566105.39       919415.29
      1565557.39       919637.52
#Sta/Elev= 30
  4654.1  807.23  4691.7  800.34  4708.3  795.75  4724.8  792.10  4745.2  786.57
  4755.8  782.75  4799.7  769.73  4811.0  765.63  4828.9  766.88  4868.4  767.04
  4888.4  767.57  4916.7  766.85  4944.0  767.64  4984.3  763.53  4987.3  758.53
  5012.7  758.53  5015.7  763.53  5030.4  767.80  5042.7  767.44  5104.0  767.00
  5117.4  766.49  5186.9  768.05  5203.6  767.47  5214.1  767.58  5221.8  767.99
  5263.1  786.37  5292.5  794.79  5306.3  797.77  5319.9  801.23  5360.2  808.35
#Mann=5,-1,0
  4654.1    0.13       0  4984.3    0.05       0  5015.7    0.13       0
  5042.7    0.07       0  5214.1    0.13       0
#XS Ineff=2,0
    0.00 4860.60  779.08 5139.40    0.00  779.08
Permanent Ineff=
       F       F
Bank Sta=4984.3,5015.7
XS Rating Curve= 0
Exp/Cntr=0.3,0.1

Type RM Length L Ch R = 1,4081,250,250,250
BEGIN DESCRIPTION:
Grassy Creek 9.0
END DESCRIPTION:
XS GIS Cut Line= 3
      1566072.53       919112.26      1565900.84       919152.66
      1565815.06       919145.09
#Sta/Elev= 30
  4909.4  800.95  4913.8  799.90  4922.4  793.12  4933.8  786.50  4949.3  776.64
  4962.5  768.58  4966.6  767.26  4983.9  760.89  4986.9  755.89  5013.1  755.89
  5016.1  760.89  5024.4  761.77  5029.2  764.05  5034.6  763.63  5044.8  763.73
  5058.2  766.50  5066.4  769.12  5069.0  769.72  5088.2  775.90  5100.6  778.91
  5105.5  781.37  5113.2  783.77  5117.5  785.37  5127.2  788.16  5133.4  789.71
  5138.5  791.27  5145.7  792.95  5152.0  794.79  5161.8  797.02  5171.9  798.82
#Mann=3,-1,0
  4909.4    0.13       0  4983.9    0.05       0  5016.1    0.13       0
Bank Sta=4983.9,5016.1
XS Rating Curve= 0
Exp/Cntr=0.3,0.1

Type RM Length L Ch R = 1,3831,276,276,276
BEGIN DESCRIPTION:
Grassy Creek 8.0
END DESCRIPTION:
XS GIS Cut Line= 2
      1565981.66       918864.76      1565761.93       918955.69
#Sta/Elev= 24
  4889.5  787.42  4897.4  785.86  4915.1  781.37  4932.1  775.86  4942.8  772.03
  4947.7  770.52  4953.5  769.27  4971.0  764.91  4974.7  763.69  4983.9  760.06
  4986.9  755.06  5013.1  755.06  5016.1  760.06  5025.9  763.46  5026.3  763.47
  5027.8  763.64  5042.2  764.84  5060.7  769.48  5069.0  771.11  5092.5  776.44
  5103.0  779.74  5103.9  780.09  5122.4  785.59  5127.3  787.21
#Mann=3,-1,0
  4889.5    0.13       0  4983.9    0.05       0  5016.1    0.13       0
Bank Sta=4983.9,5016.1
XS Rating Curve= 0
Exp/Cntr=0.3,0.1

Type RM Length L Ch R = 1,3555,301,301,301
BEGIN DESCRIPTION:
Grassy Creek 7.0
END DESCRIPTION:
XS GIS Cut Line= 2
      1565931.16       918624.86      1565673.59       918672.84
#Sta/Elev= 30
  4837.3  789.02  4853.2  786.57  4864.2  784.02  4871.4  783.06  4877.6  781.47
  4885.9  778.03  4891.2  776.13  4897.5  774.16  4901.0  773.27  4903.9  772.31
  4910.9  770.44  4921.5  767.98  4936.0  767.35  4949.6  765.89  4952.5  765.67
  4962.7  765.37  4975.9  761.87  4983.6  760.48  4983.9  759.63  4986.9  754.63
  5013.1  754.63  5016.1  759.63  5021.9  761.08  5032.0  765.33  5036.9  766.90
  5047.8  771.05  5060.9  775.49  5075.3  780.05  5088.6  783.74  5099.3  787.50
#Mann=3,-1,0
  4837.3    0.13       0  4983.9    0.05       0  5016.1    0.13       0
Bank Sta=4983.9,5016.1
XS Rating Curve= 0
Exp/Cntr=0.3,0.1

Type RM Length L Ch R = 1,3254,249,249,249
BEGIN DESCRIPTION:
Grassy Creek 6.0
END DESCRIPTION:
XS GIS Cut Line= 2
      1566001.86       918541.54      1565873.04       918352.09
#Sta/Elev= 26
  4861.4  783.25  4868.3  781.88  4881.7  778.33  4885.5  777.11  4891.1  775.41
  4906.5  771.34  4909.1  770.85  4926.0  768.18  4933.3  766.77  4936.9  766.31
  4938.6  766.12  4958.4  764.53  4963.4  764.44  4965.9  764.50  4971.8  761.96
  4977.6  759.83  4982.1  758.44  4983.9  758.13  4986.9  753.13  5013.1  753.13
  5016.1  758.13  5028.6  767.78  5058.5  783.40  5065.7  787.58  5080.5  795.49
  5090.5  800.00
#Mann=3,-1,0
  4861.4    0.13       0  4983.9    0.05       0  5016.1    0.13       0
Bank Sta=4983.9,5016.1
XS Rating Curve= 0
Exp/Cntr=0.3,0.1

Type RM Length L Ch R = 1,3005,204,204,204
BEGIN DESCRIPTION:
Grassy Creek 5.0
END DESCRIPTION:
XS GIS Cut Line= 3
      1566208.93       918480.92      1566196.31       918400.11
      1566110.44       918256.16
#Sta/Elev= 25
  4825.3  781.37  4830.6  780.67  4837.2  779.95  4863.1  776.08  4879.3  774.61
  4882.7  774.21  4888.8  772.91  4907.1  769.68  4934.0  765.83  4948.8  763.06
  4954.3  762.97  4958.8  762.64  4962.4  762.62  4977.4  760.51  4978.4  760.43
  4979.2  760.16  4983.9  757.78  4986.9  752.78  5013.1  752.78  5016.1  757.78
  5037.1  769.47  5041.0  770.63  5049.4  775.26  5058.3  780.96  5074.7  789.71
#Mann=3,-1,0
  4825.3    0.13       0  4983.9    0.05       0  5016.1    0.13       0
Bank Sta=4983.9,5016.1
XS Rating Curve= 0
Exp/Cntr=0.3,0.1

Type RM Length L Ch R = 1,2801,208,208,208
BEGIN DESCRIPTION:
Grassy Creek 4.0
END DESCRIPTION:
XS GIS Cut Line= 2
      1566380.66       918283.95      1566274.60       918157.68
#Sta/Elev= 15
  4914.8  784.96  4930.2  778.82  4932.8  778.01  4951.2  766.12  4960.7  763.30
  4974.6  758.70  4982.6  757.29  4985.8  752.29  5014.2  752.29  5017.4  757.29
  5039.0  761.09  5039.6  761.27  5040.2  761.58  5041.2  761.94  5079.7  779.51
#Mann=3,-1,0
  4914.8    0.13       0  4982.6    0.05       0  5017.4    0.13       0
Bank Sta=4982.6,5017.4
XS Rating Curve= 0
Exp/Cntr=0.3,0.1

Type RM Length L Ch R = 1,2593,160,160,160
BEGIN DESCRIPTION:
Grassy Creek 3.0
END DESCRIPTION:
XS GIS Cut Line= 3
      1566587.71       918132.42      1566532.17       918117.27
      1566375.70       918021.36
#Sta/Elev= 30
  4892.3  793.56  4906.1  786.12  4913.3  780.57  4926.8  771.62  4930.8  768.58
  4941.0  762.46  4946.8  760.84  4950.1  759.63  4969.7  755.24  4974.0  750.24
  5000.0  750.24  5004.3  755.24  5009.0  758.31  5011.9  759.00  5014.8  759.48
  5024.4  761.72  5045.1  764.17  5053.6  764.71  5060.1  766.46  5065.4  767.36
  5070.2  769.77  5073.2  771.08  5085.3  775.44  5091.3  776.02  5093.2  776.44
  5104.6  780.77  5106.6  781.35  5113.7  784.20  5125.5  787.62  5133.4  790.62
#Mann=3,-1,0
  4892.3    0.13       0  4969.7    0.05       0  5004.3    0.13       0
Bank Sta=4969.7,5004.3
XS Rating Curve= 0
Exp/Cntr=0.3,0.1

Type RM Length L Ch R = 1,2433,210,210,210
BEGIN DESCRIPTION:
Grassy Creek 2.0
END DESCRIPTION:
XS GIS Cut Line= 3
      1566696.28       918038.96      1566493.03       917903.88
      1566429.89       917910.20
#Sta/Elev= 30
  4877.8  798.31  4894.3  792.95  4899.5  791.06  4915.4  784.54  4924.3  781.82
  4937.4  777.28  4945.3  771.90  4962.2  761.85  4966.0  759.89  4981.7  756.28
  4982.6  754.44  4985.8  749.44  5014.2  749.44  5017.4  754.44  5024.4  754.97
  5027.2  756.62  5032.5  757.87  5038.9  759.93  5060.0  761.32  5067.4  762.95
  5079.7  767.13  5087.4  769.02  5096.0  769.70  5098.8  770.56  5110.0  772.13
  5119.6  774.08  5136.0  775.85  5149.5  778.68  5163.4  780.07  5185.3  782.96
#Mann=3,-1,0
  4877.8    0.13       0  4982.6    0.05       0  5017.4    0.13       0
Bank Sta=4982.6,5017.4
XS Rating Curve= 0
Exp/Cntr=0.5,0.3

Type RM Length L Ch R = 1,2223,106,106,106
BEGIN DESCRIPTION:
Railroad (GC) us
END DESCRIPTION:
XS GIS Cut Line= 5
      1567017.19       917751.97      1566858.96       917779.30
      1566630.29       917828.20      1566538.25       917854.09
      1566401.60       917895.80
#Sta/Elev= 30
  4702.8  801.95  4710.0  801.07  4751.6  789.66  4774.0  781.23  4793.4  777.37
  4806.0  773.41  4813.2  773.46  4825.0  769.71  4834.4  768.10  4841.6  765.07
  4864.1  762.21  4885.1  761.57  4912.9  759.01  4935.2  758.13  4970.0  753.87
  4985.0  748.87  5015.0  748.87  5030.0  753.87  5045.5  757.90  5057.9  758.16
  5111.0  768.90  5155.8  772.68  5167.3  772.50  5194.9  774.00  5218.8  771.95
  5232.8  771.60  5266.1  777.01  5290.9  778.84  5310.2  783.75  5335.7  787.21
#Mann=3,-1,0
  4702.8    0.13       0  4970.0    0.05       0  5030.0    0.13       0
#XS Ineff=2,0
    0.00 4886.00  769.22 5114.00    0.00  769.64
Permanent Ineff=
       F       F
Bank Sta=4970,5030
XS Rating Curve= 0
Exp/Cntr=0.5,0.3

Type RM Length L Ch R =3,2167,,,
BEGIN DESCRIPTION:
Railroad (GC) TOR
Structure ID: GC_RR_estimate
Approximate Survey Structure
END DESCRIPTION:
Bridge Culvert--1,0,-1,-1,0
Deck Dist Width WeirC Skew NumUp NumDn MinLoCord MaxHiCord MaxSubmerge Is_Ogee
49,14,3,,17,17,,,0.95,0,1,1,,,
  4726.5  4742.1  4786.4  4806.4  4837.9  4891.1  4935.0  4935.0  5065.0  5065.0
  5151.8  5215.3  5287.1  5332.5  5380.0  5394.0  5452.3
  796.95  792.89  774.57  770.21  769.57  769.09  768.70  768.70  768.70  768.70
  770.09  770.21  770.60  774.77  784.92  787.48  790.01
  728.87  728.87  728.87  728.87  728.87  728.87  728.87  767.20  767.20  728.87
  728.87  728.87  728.87  728.87  728.87  728.87  728.87
  4726.5  4742.1  4786.4  4806.4  4837.9  4891.1  4935.0  4935.0  5065.0  5065.0
  5151.8  5215.3  5287.1  5332.5  5380.0  5394.0  5452.3
  796.95  792.89  774.57  770.21  769.57  769.09  768.70  768.70  768.70  768.70
  770.09  770.21  770.60  774.77  784.92  787.48  790.01
  728.87  728.87  728.87  728.87  728.87  728.87  728.87  767.20  767.20  728.87
  728.87  728.87  728.87  728.87  728.87  728.87  728.87
Pier Skew, UpSta & Num, DnSta & Num=,4956.7,2,4956.7,2,0,0,0,0,0
       1       1
  748.00  767.20
       1       1
  748.00  767.20
Pier Skew, UpSta & Num, DnSta & Num=,5000,2,5000,2,0,0,0,0,0
       1       1
  748.00  767.20
       1       1
  748.00  767.20
Pier Skew, UpSta & Num, DnSta & Num=,5043.3,2,5043.3,2,0,0,0,0,0
       1       1
  748.00  767.20
       1       1
  748.00  767.20
Abutment Skew #Up #Dn=,2,2
  4935.0  4940.0
  767.20  757.52
  4935.0  4940.0
  767.20  761.44
Abutment Skew #Up #Dn=,2,2
  5060.0  5065.0
  758.63  767.20
  5060.0  5065.0
  760.54  767.20
BR Coef=1,1,0,1.25,0,,,0.8,0,2,0,
WSPro=,,,, 1 ,,,, 0 ,,,, 0 ,,,,-1 ,-1 ,-1 , 0 , 0 , 0 , 0 , 0
BC Design=,,0,,0,,,,,,

Type RM Length L Ch R = 1,2117,65,65,65
BEGIN DESCRIPTION:
Railroad (GC) ds
END DESCRIPTION:
XS GIS Cut Line= 5
      1567027.19       917731.83      1566939.49       917688.70
      1566617.35       917760.61      1566473.54       917790.81
      1566384.36       917888.61
#Sta/Elev= 30
  4746.9  794.37  4754.6  791.36  4783.6  775.41  4797.3  769.81  4819.0  768.36
  4842.0  761.42  4869.4  761.87  4889.6  764.20  4897.6  760.15  4927.5  763.89
  4937.1  762.43  4948.2  758.63  4964.5  756.05  4970.0  753.62  4985.0  748.62
  5015.0  748.62  5030.0  753.62  5054.6  760.72  5082.1  760.87  5173.2  759.35
  5185.2  760.71  5206.1  759.45  5258.0  761.15  5280.2  760.28  5301.8  761.65
  5324.4  761.70  5359.1  768.30  5412.4  771.28  5428.3  780.95  5454.0  786.85
#Mann=5,-1,0
  4746.9    0.13       0  4970.0    0.05       0  5030.0    0.13       0
  5082.1    0.07       0  5301.8    0.13       0
#XS Ineff=2,0
    0.00 4892.00  769.12 5108.00    0.00  769.90
Permanent Ineff=
       F       F
Bank Sta=4970,5030
XS Rating Curve= 0
Exp/Cntr=0.5,0.3

Type RM Length L Ch R = 1,2052,0,0,0
BEGIN DESCRIPTION:
Grassy Creek 1.0
END DESCRIPTION:
XS GIS Cut Line= 5
      1567074.66       917714.58      1566969.69       917636.93
      1566696.45       917681.51      1566463.47       917772.11
      1566375.75       917877.08
#Sta/Elev= 30
  4711.6  793.17  4728.7  785.73  4741.9  773.98  4749.2  770.40  4769.9  768.98
  4812.2  757.70  4853.2  757.21  4916.2  760.73  4935.7  759.00  4941.0  757.64
  4974.5  753.26  4979.3  748.26  5020.7  748.26  5025.5  753.26  5040.1  755.17
  5060.6  757.85  5076.8  758.17  5203.3  757.31  5226.6  756.30  5242.4  757.13
  5266.4  756.09  5278.8  757.23  5369.0  759.24  5394.6  761.25  5414.1  766.01
  5446.2  770.05  5461.3  771.22  5477.0  770.86  5494.1  781.29  5505.8  784.05
#Mann=5,-1,0
  4711.6    0.13       0  4974.5    0.05       0  5025.5    0.13       0
  5040.1    0.07       0  5394.6    0.13       0
#XS Ineff=2,0
    0.00 4917.10  764.83 5082.90    0.00  764.83
Permanent Ineff=
       F       F
Bank Sta=4974.5,5025.5
XS Rating Curve= 0
Exp/Cntr=0.3,0.1

Chan Stop Cuts=-1
