HEC-RAS study Fisher River.prj: Fisher River Limited Detail Study

--- Fisher River.g01 (geometry) --- (continued)

Type RM Length L Ch R = 1,218994,50,50,50
BEGIN DESCRIPTION:
Off Lumber Plant Rd (2) - US
END DESCRIPTION:
XS GIS Cut Line= 5
      1450823.54      1021716.18      1450693.67      1021677.03
      1450656.04      1021723.69      1450648.52      1021898.68
      1450543.18      1022037.88
#Sta/Elev= 30
  4825.0 1450.11  4838.6 1447.11  4847.7 1445.51  4877.9 1437.77  4882.8 1437.25
  4899.5 1437.03  4937.0 1432.57  4952.5 1430.41  4956.1 1429.37  4966.9 1427.30
  4972.9 1426.75  4993.7 1422.90  4996.2 1419.40  5003.9 1419.40  5006.3 1422.90
  5010.6 1425.48  5016.9 1423.95  5026.7 1425.36  5044.1 1425.81  5098.7 1428.29
  5179.3 1432.85  5220.4 1434.61  5250.6 1436.75  5267.0 1438.93  5278.0 1440.83
  5297.5 1442.78  5305.6 1444.18  5322.4 1446.30  5359.0 1453.28  5370.3 1454.76
#Mann=4,-1,0
  4825.0    0.08       0  4937.0    0.14       0  4993.7    0.04       0
  5006.3    0.08       0
#XS Ineff=2,0
    0.00 4982.00 1427.50 5018.00    0.00 1427.50
Permanent Ineff=
       F       F
Bank Sta=4993.7,5006.3
XS Rating Curve= 0
Exp/Cntr=0.5,0.3

Type RM Length L Ch R =3,218966,,,
BEGIN DESCRIPTION:
Off Lumber Plant Rd (2) - TOR
Structure ID: LDS_FR_25B
Approximate Survey Structure
END DESCRIPTION:
Bridge Culvert--1,0,-1,-1,0
Deck Dist Width WeirC Skew NumUp NumDn MinLoCord MaxHiCord MaxSubmerge Is_Ogee
22,12,3,,49,49,,,0.95,0,1,1,,,
  4769.7  4800.0  4806.9  4809.2  4811.6  4823.6  4864.0  4885.5  4910.6  4963.9
  4992.5  4992.5  5007.5  5007.5  5105.1  5106.2  5113.6  5125.3  5125.8  5126.2
  5141.0  5155.1  5156.6  5171.5  5183.9  5186.0  5186.5  5201.0  5206.5  5223.8
  5226.1  5238.6  5241.8  5242.7  5245.3  5260.1  5268.3  5270.1  5281.8  5284.2
  5302.7  5306.9  5312.0  5325.6  5331.6  5343.9  5352.5  5355.8  5374.7
 1456.33 1450.59 1448.92 1448.47 1448.13 1445.45 1436.14 1433.28 1430.77 1427.50
 1427.50 1427.50 1427.50 1427.50 1427.50 1427.56 1427.81 1428.76 1428.79 1428.80
 1428.69 1430.17 1430.27 1430.77 1431.96 1432.13 1432.18 1432.65 1433.02 1433.89
 1433.96 1434.62 1435.13 1435.18 1435.57 1436.12 1436.69 1436.96 1438.27 1438.48
 1440.62 1440.99 1441.59 1443.39 1444.26 1445.75 1447.44 1447.91 1451.29
 1399.40 1399.40 1399.40 1399.40 1399.40 1399.40 1399.40 1399.40 1399.40 1399.40
 1399.40 1425.50 1425.50 1399.40 1399.40 1399.40 1399.40 1399.40 1399.40 1399.40
 1399.40 1399.40 1399.40 1399.40 1399.40 1399.40 1399.40 1399.40 1399.40 1399.40
 1399.40 1399.40 1399.40 1399.40 1399.40 1399.40 1399.40 1399.40 1399.40 1399.40
 1399.40 1399.40 1399.40 1399.40 1399.40 1399.40 1399.40 1399.40 1399.40
  4769.7  4800.0  4806.9  4809.2  4811.6  4823.6  4864.0  4885.5  4910.6  4963.9
  4992.5  4992.5  5007.5  5007.5  5105.1  5106.2  5113.6  5125.3  5125.8  5126.2
  5141.0  5155.1  5156.6  5171.5  5183.9  5186.0  5186.5  5201.0  5206.5  5223.8
  5226.1  5238.6  5241.8  5242.7  5245.3  5260.1  5268.3  5270.1  5281.8  5284.2
  5302.7  5306.9  5312.0  5325.6  5331.6  5343.9  5352.5  5355.8  5374.7
 1456.33 1450.59 1448.92 1448.47 1448.13 1445.45 1436.14 1433.28 1430.77 1427.50
 1427.50 1427.50 1427.50 1427.50 1427.50 1427.56 1427.81 1428.76 1428.79 1428.80
 1428.69 1430.17 1430.27 1430.77 1431.96 1432.13 1432.18 1432.65 1433.02 1433.89
 1433.96 1434.62 1435.13 1435.18 1435.57 1436.12 1436.69 1436.96 1438.27 1438.48
 1440.62 1440.99 1441.59 1443.39 1444.26 1445.75 1447.44 1447.91 1451.29
 1399.40 1399.40 1399.40 1399.40 1399.40 1399.40 1399.40 1399.40 1399.40 1399.40
 1399.40 1425.50 1425.50 1399.40 1399.40 1399.40 1399.40 1399.40 1399.40 1399.40
 1399.40 1399.40 1399.40 1399.40 1399.40 1399.40 1399.40 1399.40 1399.40 1399.40
 1399.40 1399.40 1399.40 1399.40 1399.40 1399.40 1399.40 1399.40 1399.40 1399.40
 1399.40 1399.40 1399.40 1399.40 1399.40 1399.40 1399.40 1399.40 1399.40
Abutment Skew #Up #Dn=,2,2
  4992.5  4994.0
 1425.50 1421.19
  4992.5  4994.0
 1425.50 1420.94
Abutment Skew #Up #Dn=,2,2
  5006.0  5007.5
 1421.19 1425.50
  5006.0  5007.5
 1420.94 1425.50
BR Coef=1,1,0,1.25,0,,,0.8,0,2,0,
WSPro=,,,, 1 ,,,, 0 ,,,, 0 ,,,,-1 ,-1 ,-1 , 0 , 0 , 0 , 0 , 0
BC Design=,,0,,0,,,,,,

Type RM Length L Ch R = 1,218944,224,224,224
BEGIN DESCRIPTION:
Off Lumber Plant Rd (2) - DS
END DESCRIPTION:
XS GIS Cut Line= 4
      1450840.40      1021682.67      1450674.86      1021628.11
      1450501.76      1021829.44      1450403.91      1021872.71
#Sta/Elev= 30
  4769.5 1451.25  4775.8 1450.06  4792.1 1445.79  4812.1 1442.38  4835.9 1437.02
  4841.0 1436.41  4861.5 1431.12  4900.9 1427.81  4915.0 1427.05  4954.6 1426.35
  4979.7 1424.24  4985.7 1423.25  4993.7 1422.65  4996.2 1419.15  5003.9 1419.15
  5006.3 1422.65  5011.0 1423.94  5018.9 1424.97  5047.1 1425.61  5088.7 1427.33
  5129.5 1430.05  5157.0 1432.11  5184.1 1433.37  5197.0 1435.47  5223.0 1442.05
  5249.4 1450.91  5262.7 1454.44  5290.2 1460.05  5299.0 1461.43  5316.3 1463.29
#Mann=4,-1,0
  4769.5    0.08       0  4993.7    0.04       0  5006.3    0.14       0
  5129.5    0.08       0
#XS Ineff=2,0
    0.00 4982.00 1426.00 5018.00    0.00 1426.00
Permanent Ineff=
       F       F
Bank Sta=4993.7,5006.3
XS Rating Curve= 0
Exp/Cntr=0.5,0.3

Type RM Length L Ch R = 1,218720,464,464,464
BEGIN DESCRIPTION:
Fisher River 437.0
END DESCRIPTION:
XS GIS Cut Line= 3
      1450906.33      1021460.66      1450563.85      1021453.13
      1450304.21      1021618.70
#Sta/Elev= 30
  4616.1 1452.14  4625.9 1449.20  4637.4 1444.00  4656.6 1437.51  4682.1 1430.65
  4687.5 1428.73  4691.0 1428.36  4704.9 1427.67  4723.2 1426.16  4746.6 1425.23
  4795.2 1422.19  4811.4 1421.85  4867.3 1422.17  4896.3 1421.59  4936.4 1421.68
  4979.7 1422.59  4990.2 1422.22  4998.5 1418.87  5000.8 1413.87  5007.5 1413.87
  5009.0 1418.87  5011.5 1422.59  5014.9 1422.39  5064.9 1423.97  5106.4 1427.59
  5140.2 1435.67  5187.5 1449.80  5226.0 1459.52  5238.9 1462.46  5266.6 1464.94
#Mann=3,-1,0
  4616.1    0.08       0  4998.5    0.04       0  5009.0    0.08       0
#XS Ineff=2,0
    0.00 4903.70 1426.64               0
Permanent Ineff=
       F       F
Bank Sta=4998.5,5009
XS Rating Curve= 0
Exp/Cntr=0.5,0.3

Type RM Length L Ch R = 1,218256,54,54,54
BEGIN DESCRIPTION:
Lumber Plant Rd - US
END DESCRIPTION:
XS GIS Cut Line= 4
      1450904.43      1021452.38      1450689.91      1021444.85
      1450418.97      1021053.49      1450371.96      1021030.92
#Sta/Elev= 30
  4333.1 1451.49  4342.1 1448.87  4360.5 1440.86  4374.6 1436.60  4394.0 1429.65
  4405.7 1428.26  4435.8 1426.20  4486.9 1423.09  4512.6 1421.99  4539.5 1421.49
  4570.8 1421.62  4716.3 1419.32  4776.0 1418.15  4796.4 1417.19  4820.6 1416.69
  4849.9 1417.22  4952.9 1415.22  4981.6 1411.61  4990.8 1411.20  4994.0 1407.80
  5006.0 1407.80  5009.2 1411.20  5010.9 1411.46  5011.5 1410.95  5020.9 1412.76
  5023.8 1414.94  5047.8 1440.92  5056.2 1445.67  5059.7 1448.10  5075.9 1455.95
#Mann=3,-1,0
  4333.1    0.08       0  4990.8    0.04       0  5009.2    0.14       0
#XS Ineff=2,0
    0.00 4965.00 1418.40 5035.00    0.00 1418.40
Permanent Ineff=
       F       F
Bank Sta=4990.8,5009.2
XS Rating Curve= 0
Exp/Cntr=0.5,0.3

Type RM Length L Ch R =3,218235,,,
BEGIN DESCRIPTION:
Lumber Plant Rd - TOR
Structure ID: LDS_FR_25A
Approximate Survey Structure
END DESCRIPTION:
Bridge Culvert--1,0,-1,-1,0
Deck Dist Width WeirC Skew NumUp NumDn MinLoCord MaxHiCord MaxSubmerge Is_Ogee
11,20,3,,7,7,,,0.95,0,1,1,,,
  4733.8  4748.5  4985.0  4985.0  5015.0  5015.0  5037.8
 1418.50 1418.40 1418.40 1418.40 1418.40 1418.40 1418.40
 1387.80 1387.80 1387.80 1416.40 1416.40 1387.80 1387.80
  4733.8  4748.5  4985.0  4985.0  5015.0  5015.0  5037.8
 1418.50 1418.40 1418.40 1418.40 1418.40 1418.40 1418.40
 1387.80 1387.80 1387.80 1416.40 1416.40 1387.80 1387.80
BR Coef=1,1,0,1.25,0,,,0.8,0,2,0,
WSPro=,,,, 1 ,,,, 0 ,,,, 0 ,,,,-1 ,-1 ,-1 , 0 , 0 , 0 , 0 , 0
BC Design=,,0,,0,,,,,,

Type RM Length L Ch R = 1,218202,279,279,279
BEGIN DESCRIPTION:
Lumber Plant Rd - DS
END DESCRIPTION:
XS GIS Cut Line= 4
      1450898.78      1021412.87      1450742.20      1021404.75
      1450445.31      1021000.81      1450379.50      1020976.36
#Sta/Elev= 30
  4386.3 1449.69  4395.0 1447.13  4438.2 1428.97  4456.7 1426.35  4532.6 1422.94
  4616.7 1420.69  4646.0 1420.45  4703.0 1419.30  4718.4 1419.37  4738.7 1418.77
  4769.4 1418.38  4793.3 1417.81  4870.7 1414.78  4900.8 1415.01  4923.2 1414.28
  4970.3 1414.53  4988.5 1413.55  4992.5 1407.55  5007.5 1407.55  5011.5 1413.55
  5015.8 1416.57  5032.1 1418.47  5039.7 1418.71  5049.2 1417.98  5056.2 1418.31
  5059.0 1422.04  5061.9 1434.42  5083.2 1445.27  5088.3 1448.25  5114.6 1461.05
#Mann=3,-1,0
  4386.3    0.08       0  4988.5    0.04       0  5011.5    0.14       0
#XS Ineff=2,0
    0.00 4965.00 1418.00 5035.00    0.00 1418.00
Permanent Ineff=
       F       F
Bank Sta=4988.5,5011.5
XS Rating Curve= 0
Exp/Cntr=0.5,0.3

Type RM Length L Ch R = 1,217923,420,420,420
BEGIN DESCRIPTION:
Fisher River 436.0
END DESCRIPTION:
XS GIS Cut Line= 3
      1450967.96      1021282.22      1450690.64      1020886.90
      1450569.71      1020736.47
#Sta/Elev= 30
  4464.7 1453.41  4518.8 1442.11  4547.3 1433.99  4568.1 1427.20  4575.3 1425.62
  4608.7 1426.05  4645.3 1425.04  4686.5 1421.08  4730.3 1419.36  4777.8 1416.34
  4831.3 1415.14  4901.9 1412.79  4942.6 1412.16  4971.6 1412.20  4984.9 1413.08
  4988.4 1412.63  4990.7 1413.29  4994.3 1407.57  4996.8 1402.57  5003.2 1402.57
  5005.7 1407.57  5006.0 1409.46  5008.4 1409.55  5015.4 1413.94  5023.1 1414.62
  5040.3 1414.54  5062.0 1424.09  5082.1 1431.06  5093.0 1435.56  5140.6 1446.39
#Mann=3,-1,0
  4464.7    0.08       0  4994.3    0.04       0  5005.7    0.14       0
Bank Sta=4994.3,5005.7
XS Rating Curve= 0
Exp/Cntr=0.3,0.1

Type RM Length L Ch R = 1,217503,493,493,493
BEGIN DESCRIPTION:
Fisher River 435.0
END DESCRIPTION:
XS GIS Cut Line= 3
      1451097.80      1020624.35      1450876.50      1020544.68
      1450690.61      1020432.55
#Sta/Elev= 30
  4847.3 1458.75  4860.2 1453.35  4883.1 1440.54  4909.8 1425.03  4918.3 1419.19
  4922.5 1417.56  4937.9 1413.40  4969.6 1407.22  4985.5 1403.03  4994.3 1402.65
  4996.8 1396.95  5003.2 1396.95  5005.7 1402.65  5011.5 1404.74  5022.0 1407.77
  5045.5 1408.36  5117.0 1408.06  5164.4 1408.38  5176.1 1409.52  5181.2 1410.72
  5185.1 1412.97  5188.9 1415.25  5205.3 1417.13  5214.3 1417.08  5219.8 1420.51
  5234.8 1427.59  5238.9 1428.29  5265.6 1437.86  5290.7 1445.25  5299.6 1448.29
#Mann=5,-1,0
  4847.3    0.14       0  4937.9    0.08       0  4994.3    0.04       0
  5005.7    0.08       0  5185.1    0.14       0
#XS Ineff=2,0
       0                 5045.50    0.00 1408.36
Permanent Ineff=
       F       F
Bank Sta=4994.3,5005.7
XS Rating Curve= 0
Exp/Cntr=0.3,0.1

Type RM Length L Ch R = 1,217010,393,393,393
BEGIN DESCRIPTION:
Fisher River 434.0
END DESCRIPTION:
XS GIS Cut Line= 3
      1450982.67      1020109.54      1450900.10      1020106.59
      1450637.51      1020192.15
#Sta/Elev= 30
  4851.3 1451.12  4876.2 1442.67  4879.1 1441.52  4889.5 1436.82  4901.1 1432.98
  4950.5 1410.51  4955.3 1407.98  4969.1 1401.68  4984.9 1397.29  4994.3 1395.94
  4996.8 1390.94  5003.2 1390.94  5005.7 1395.94  5011.3 1396.94  5019.1 1400.67
  5021.5 1403.45  5032.6 1408.87  5039.4 1410.04  5052.8 1410.80  5061.2 1419.96
  5064.2 1423.56  5092.7 1435.13  5106.3 1437.86  5110.9 1439.04  5121.7 1442.38
  5133.7 1444.64  5161.1 1450.76  5182.0 1455.08  5202.5 1458.42  5210.1 1459.89
#Mann=3,-1,0
  4851.3    0.14       0  4994.3    0.04       0  5005.7    0.14       0
Bank Sta=4994.3,5005.7
XS Rating Curve= 0
Exp/Cntr=0.3,0.1

Type RM Length L Ch R = 1,216617,370,370,370
BEGIN DESCRIPTION:
Fisher River 433.0
END DESCRIPTION:
XS GIS Cut Line= 4
      1451026.99      1019873.55      1450878.60      1019770.39
      1450761.45      1019737.82      1450649.34      1019950.23
#Sta/Elev= 30
  4776.7 1452.41  4806.7 1443.09  4832.1 1432.74  4849.2 1425.02  4858.4 1421.82
  4874.2 1415.07  4906.6 1402.97  4932.9 1393.87  4965.4 1393.21  4994.3 1389.78
  4996.8 1384.78  5003.2 1384.78  5005.7 1389.78  5022.2 1392.55  5027.7 1394.07
  5032.2 1394.64  5034.5 1394.19  5049.8 1394.43  5074.9 1398.06  5079.0 1399.24
  5089.1 1398.06  5109.7 1401.36  5133.2 1403.05  5170.7 1404.63  5187.9 1406.28
  5237.0 1412.28  5251.9 1414.95  5265.1 1416.06  5288.0 1420.20  5319.2 1424.63
#Mann=3,-1,0
  4776.7    0.14       0  4994.3    0.04       0  5005.7    0.08       0
Bank Sta=4994.3,5005.7
XS Rating Curve= 0
Exp/Cntr=0.5,0.3

Type RM Length L Ch R = 1,216247,56,56,56
BEGIN DESCRIPTION:
Off Lumber Plant Rd - US
END DESCRIPTION:
XS GIS Cut Line= 4
      1451239.36      1019652.25      1451156.77      1019507.71
      1450696.55      1019330.70      1450634.62      1019318.91
#Sta/Elev= 30
  4708.3 1430.01  4755.4 1414.49  4780.3 1407.49  4836.0 1396.47  4867.4 1393.32
  4886.1 1392.27  4942.4 1390.61  4956.9 1390.74  4966.5 1392.02  4987.0 1386.45
  4991.3 1385.91  4995.5 1379.81  5004.5 1379.81  5008.8 1385.91  5013.8 1388.54
  5028.9 1387.36  5044.4 1387.27  5148.4 1389.63  5173.1 1392.69  5179.0 1395.50
  5196.2 1398.31  5236.8 1399.01  5245.3 1400.34  5255.7 1405.06  5258.9 1405.85
  5292.4 1407.87  5350.6 1414.52  5371.5 1419.10  5418.7 1423.17  5430.9 1426.63
#Mann=3,-1,0
  4708.3    0.14       0  4991.3    0.04       0  5008.8    0.08       0
#XS Ineff=2,0
    0.00 4974.00 1390.15 5026.00    0.00 1390.15
Permanent Ineff=
       F       F
Bank Sta=4991.3,5008.8
XS Rating Curve= 0
Exp/Cntr=0.5,0.3

Type RM Length L Ch R =3,216220,,,
BEGIN DESCRIPTION:
Off Lumber Plant Rd - TOR
Structure ID: LDS_FR_25
Approximate Survey Structure
END DESCRIPTION:
Bridge Culvert--1,0,-1,-1,0
Deck Dist Width WeirC Skew NumUp NumDn MinLoCord MaxHiCord MaxSubmerge Is_Ogee
21.5,11,3,,29,29,,,0.95,0,1,1,,,
  4770.8  4784.3  4786.0  4793.4  4827.2  4852.9  4860.1  4885.6  4901.3  4916.6
  4925.5  4949.1  4949.6  4959.3  4984.0  4984.0  5016.0  5016.0  5124.2  5124.8
  5138.8  5146.0  5162.1  5182.0  5182.5  5191.2  5204.0  5205.0  5212.2
 1407.31 1404.98 1404.65 1403.44 1397.74 1394.71 1393.97 1392.36 1391.67 1391.13
 1390.71 1390.38 1390.40 1390.11 1390.10 1390.10 1390.10 1390.10 1390.43 1390.42
 1390.97 1391.53 1393.23 1396.11 1396.19 1397.19 1398.18 1398.23 1398.35
 1359.81 1359.81 1359.81 1359.81 1359.81 1359.81 1359.81 1359.81 1359.81 1359.81
 1359.81 1359.81 1359.81 1359.81 1359.81 1388.60 1388.60 1359.81 1359.81 1359.81
 1359.81 1359.81 1359.81 1359.81 1359.81 1359.81 1359.81 1359.81 1359.81
  4770.8  4784.3  4786.0  4793.4  4827.2  4852.9  4860.1  4885.6  4901.3  4916.6
  4925.5  4949.1  4949.6  4959.3  4984.0  4984.0  5016.0  5016.0  5124.2  5124.8
  5138.8  5146.0  5162.1  5182.0  5182.5  5191.2  5204.0  5205.0  5212.2
 1407.31 1404.98 1404.65 1403.44 1397.74 1394.71 1393.97 1392.36 1391.67 1391.13
 1390.71 1390.38 1390.40 1390.11 1390.10 1390.10 1390.10 1390.10 1390.43 1390.42
 1390.97 1391.53 1393.23 1396.11 1396.19 1397.19 1398.18 1398.23 1398.35
 1359.81 1359.81 1359.81 1359.81 1359.81 1359.81 1359.81 1359.81 1359.81 1359.81
 1359.81 1359.81 1359.81 1359.81 1359.81 1388.60 1388.60 1359.81 1359.81 1359.81
 1359.81 1359.81 1359.81 1359.81 1359.81 1359.81 1359.81 1359.81 1359.81
Abutment Skew #Up #Dn=,2,2
  4984.0  4987.5
 1388.60 1385.41
  4984.0  4987.5
 1388.60 1385.16
Abutment Skew #Up #Dn=,2,2
  5012.5  5016.0
 1385.41 1388.60
  5012.5  5016.0
 1385.16 1388.60
BR Coef=1,1,0,1.25,0,,,0.8,0,2,0,
WSPro=,,,, 1 ,,,, 0 ,,,, 0 ,,,,-1 ,-1 ,-1 , 0 , 0 , 0 , 0 , 0
BC Design=,,0,,0,,,,,,

Type RM Length L Ch R = 1,216191,300,300,300
BEGIN DESCRIPTION:
Off Lumber Plant Rd - DS
END DESCRIPTION:
XS GIS Cut Line= 3
      1451319.04      1019581.48      1451195.12      1019466.41
      1450669.98      1019251.04
#Sta/Elev= 30
  4690.2 1432.52  4727.4 1422.59  4754.7 1412.75  4767.3 1408.69  4777.5 1406.20
  4818.4 1398.11  4836.4 1395.35  4865.8 1392.56  4966.4 1389.02  4979.0 1387.58
  4991.3 1384.66  4995.5 1379.56  5004.5 1379.56  5008.8 1384.66  5011.3 1386.96
  5012.2 1387.10  5052.7 1386.31  5088.4 1386.70  5171.0 1391.85  5191.1 1395.88
  5209.6 1398.31  5242.7 1399.72  5252.3 1403.06  5260.8 1405.44  5280.5 1407.20
  5312.0 1412.98  5349.8 1416.51  5362.3 1418.46  5389.0 1420.74  5426.9 1424.78
#Mann=4,-1,0
  4690.2    0.14       0  4836.4    0.08       0  4991.3    0.04       0
  5008.8    0.08       0
#XS Ineff=2,0
    0.00 4974.00 1388.40 5026.00    0.00 1388.40
Permanent Ineff=
       F       F
Bank Sta=4991.3,5008.8
XS Rating Curve= 0
Exp/Cntr=0.5,0.3

Type RM Length L Ch R = 1,215891,472,472,472
BEGIN DESCRIPTION:
Fisher River 431.0
END DESCRIPTION:
XS GIS Cut Line= 3
      1451428.16      1019442.79      1451212.82      1019147.80
      1450758.51      1019006.19
#Sta/Elev= 30
  4588.7 1425.91  4632.6 1410.99  4648.2 1404.79  4669.8 1399.27  4685.0 1394.31
  4704.9 1392.14  4733.6 1390.15  4923.2 1383.37  4972.1 1382.59  4981.1 1383.03
  4991.2 1380.55  4994.3 1378.60  4996.8 1373.60  5003.2 1373.60  5005.7 1378.60
  5021.6 1382.93  5032.1 1382.62  5068.8 1383.79  5123.1 1386.19  5144.7 1385.65
  5170.6 1390.86  5184.6 1395.26  5187.9 1395.74  5229.5 1397.20  5271.9 1401.29
  5287.5 1403.52  5313.5 1408.75  5357.0 1414.11  5391.6 1423.46  5429.8 1435.08
#Mann=4,-1,0
  4588.7    0.14       0  4669.8    0.08       0  4994.3    0.04       0
  5005.7    0.08       0
Bank Sta=4994.3,5005.7
XS Rating Curve= 0
Exp/Cntr=0.3,0.1

Type RM Length L Ch R = 1,215419,578,578,578
BEGIN DESCRIPTION:
Fisher River 430.0
END DESCRIPTION:
XS GIS Cut Line= 4
      1451646.46      1018855.73      1451528.48      1018820.33
      1451348.52      1018681.68      1451015.18      1018596.13
#Sta/Elev= 30
  4754.8 1413.63  4774.3 1399.73  4799.1 1384.11  4803.1 1382.36  4823.7 1378.24
  4915.7 1378.70  4987.3 1375.52  4993.1 1374.34  4994.3 1372.09  4996.8 1367.09
  5003.2 1367.09  5005.7 1372.09  5011.4 1375.71  5019.7 1379.00  5028.7 1377.76
  5063.0 1377.93  5084.9 1379.27  5179.6 1379.97  5199.1 1381.46  5206.8 1380.97
  5234.3 1382.04  5246.8 1385.12  5255.6 1385.61  5268.0 1388.42  5289.4 1389.08
  5307.7 1388.29  5324.6 1392.59  5357.4 1397.66  5385.3 1400.74  5449.3 1402.02
#Mann=3,-1,0
  4754.8    0.14       0  4994.3    0.04       0  5005.7    0.08       0
#XS Ineff=2,0
    0.00 4915.70 1378.70 5019.70    0.00 1379.00
Permanent Ineff=
       F       F
Bank Sta=4994.3,5005.7
XS Rating Curve= 0
Exp/Cntr=0.3,0.1

Type RM Length L Ch R = 1,214841,430,430,430
BEGIN DESCRIPTION:
Fisher River 429.0
END DESCRIPTION:
XS GIS Cut Line= 3
      1451879.54      1018451.56      1451696.64      1018318.81
      1451227.60      1018174.26
#Sta/Elev= 30
  4872.0 1405.78  4893.5 1406.10  4915.8 1400.44  4926.4 1401.27  4933.9 1397.80
  4946.2 1390.23  4957.6 1386.48  4969.8 1373.99  4982.4 1366.85  4994.3 1365.86
  4996.8 1360.86  5003.2 1360.86  5005.7 1365.86  5015.3 1368.30  5031.3 1369.96
  5056.6 1368.82  5129.2 1371.11  5184.1 1370.28  5243.7 1371.31  5287.7 1370.60
  5318.1 1371.62  5399.9 1372.35  5433.3 1374.16  5449.3 1378.55  5470.2 1385.80
  5478.1 1387.64  5499.7 1387.78  5514.7 1391.21  5544.9 1391.42  5588.8 1393.12
#Mann=3,-1,0
  4872.0    0.14       0  4994.3    0.04       0  5005.7    0.08       0
#XS Ineff=2,0
       0                 5131.50    0.00 1374.35
Permanent Ineff=
       F       F
Bank Sta=4994.3,5005.7
XS Rating Curve= 0
Exp/Cntr=0.5,0.3

Type RM Length L Ch R = 1,214411,103,103,103
BEGIN DESCRIPTION:
North Wilson Rd - US
END DESCRIPTION:
XS GIS Cut Line= 4
      1451879.53      1018240.60      1451773.34      1018007.57
      1451469.48      1017886.61      1451230.54      1018101.96
#Sta/Elev= 30
  4636.3 1400.20  4677.1 1391.96  4696.1 1393.07  4716.1 1391.26  4746.6 1390.92
  4791.0 1388.24  4809.9 1383.50  4813.5 1381.85  4828.8 1377.64  4888.1 1368.91
  4908.5 1367.13  4963.3 1365.13  4991.0 1360.70  4995.5 1355.10  5004.5 1355.10
  5009.0 1360.70  5022.1 1363.77  5035.9 1365.24  5108.9 1367.17  5134.7 1367.09
  5163.7 1365.39  5179.7 1366.17  5190.1 1367.58  5243.0 1371.25  5284.0 1377.15
  5357.8 1382.58  5388.7 1387.02  5423.5 1390.61  5445.5 1390.39  5541.1 1392.70
#Mann=3,-1,0
  4636.3    0.14       0  4991.0    0.04       0  5009.0    0.08       0
#XS Ineff=2,0
    0.00 4966.00 1366.90 5033.00    0.00 1366.90
Permanent Ineff=
       F       F
Bank Sta=4991,5009
XS Rating Curve= 0
Exp/Cntr=0.5,0.3

Type RM Length L Ch R =3,214362,,,
BEGIN DESCRIPTION:
North Wilson Rd - TOR
Structure ID: LDS_FR_24
Approximate Survey Structure
END DESCRIPTION:
Bridge Culvert--1,0,-1,-1,0
Deck Dist Width WeirC Skew NumUp NumDn MinLoCord MaxHiCord MaxSubmerge Is_Ogee
38.5,21,3,,19,19,,,0.95,0,1,1,,,
  4736.2  4762.5  4798.6  4808.5  4815.5  4817.9  4850.0  4879.2  4897.9  4901.5
  4910.0  4919.8  4934.3  4941.7  4977.5  4977.5  5022.5  5022.5  5188.8
 1375.70 1372.88 1371.05 1370.52 1370.26 1370.11 1368.83 1368.04 1367.50 1367.40
 1367.31 1367.12 1366.91 1366.90 1366.90 1366.90 1366.90 1366.90 1366.90
 1335.10 1335.10 1335.10 1335.10 1335.10 1335.10 1335.10 1335.10 1335.10 1335.10
 1335.10 1335.10 1335.10 1335.10 1335.10 1364.90 1364.90 1335.10 1335.10
  4736.2  4762.5  4798.6  4808.5  4815.5  4817.9  4850.0  4879.2  4897.9  4901.5
  4910.0  4919.8  4934.3  4941.7  4977.5  4977.5  5022.5  5022.5  5188.8
 1375.70 1372.88 1371.05 1370.52 1370.26 1370.11 1368.83 1368.04 1367.50 1367.40
 1367.31 1367.12 1366.91 1366.90 1366.90 1366.90 1366.90 1366.90 1366.90
 1335.10 1335.10 1335.10 1335.10 1335.10 1335.10 1335.10 1335.10 1335.10 1335.10
 1335.10 1335.10 1335.10 1335.10 1335.10 1364.90 1364.90 1335.10 1335.10
BR Coef=1,1,0,1.25,0,,,0.8,0,2,0,
WSPro=,,,, 1 ,,,, 0 ,,,, 0 ,,,,-1 ,-1 ,-1 , 0 , 0 , 0 , 0 , 0
BC Design=,,0,,0,,,,,,

Type RM Length L Ch R = 1,214308,293,293,293
BEGIN DESCRIPTION:
North Wilson Rd - DS
END DESCRIPTION:
XS GIS Cut Line= 4
      1451985.76      1017998.72      1451782.19      1017907.27
      1451454.73      1017777.46      1451168.54      1018031.20
#Sta/Elev= 30
  4662.2 1397.31  4702.4 1389.83  4737.3 1379.62  4754.9 1373.20  4771.5 1370.05
  4781.0 1367.55  4783.6 1367.66  4789.2 1366.14  4791.4 1364.73  4791.7 1365.53
  4802.6 1367.51  4822.5 1365.89  4960.9 1363.94  4982.9 1360.95  4991.1 1354.85
  5004.5 1354.85  5009.0 1360.95  5013.3 1361.90  5037.5 1363.45  5124.8 1365.45
  5183.8 1367.60  5228.6 1368.66  5299.8 1368.75  5375.9 1371.17  5431.9 1374.70
  5450.5 1378.68  5469.0 1386.29  5487.7 1388.39  5511.8 1390.26  5620.1 1394.06
#Mann=3,-1,0
  4662.2    0.14       0  4982.9    0.04       0  5009.0    0.08       0
#XS Ineff=2,0
    0.00 4956.00 1366.50 5043.00    0.00 1366.50
Permanent Ineff=
       F       F
Bank Sta=4982.9,5009
XS Rating Curve= 0
Exp/Cntr=0.5,0.3

Type RM Length L Ch R = 1,214015,425,425,425
BEGIN DESCRIPTION:
Fisher River 428.0
END DESCRIPTION:
XS GIS Cut Line= 4
      1452018.24      1017954.51      1451861.85      1017774.51
      1451855.95      1017417.54      1451425.21      1017116.62
#Sta/Elev= 30
  4691.1 1399.54  4729.4 1387.92  4764.5 1372.23  4777.2 1367.46  4786.4 1366.02
  4815.2 1363.43  4874.6 1360.86  4961.0 1362.77  4992.0 1354.00  4994.5 1348.75
  5005.5 1348.75  5008.0 1354.00  5014.3 1356.42  5034.7 1360.21  5092.8 1359.29
  5160.3 1361.37  5201.6 1357.59  5251.1 1359.78  5303.9 1359.42  5370.6 1363.31
  5520.4 1365.16  5582.8 1364.90  5596.6 1363.46  5646.8 1365.77  5701.0 1369.93
  5726.5 1375.80  5741.4 1385.94  5765.4 1398.53  5787.6 1406.09  5812.0 1411.82
#Mann=3,-1,0
  4691.1    0.14       0  4992.0    0.04       0  5008.0    0.08       0
#XS Ineff=2,0
       0                 5053.10    0.00 1360.69
Permanent Ineff=
       F       F
Bank Sta=4992,5008
XS Rating Curve= 0
Exp/Cntr=0.3,0.1

Type RM Length L Ch R = 1,213590,591,591,591
BEGIN DESCRIPTION:
Fisher River 427.0
END DESCRIPTION:
XS GIS Cut Line= 4
      1452404.67      1017733.21      1452274.87      1017585.70
      1452189.31      1017573.90      1451437.02      1017104.83
#Sta/Elev= 30
  4766.2 1387.56  4779.3 1382.38  4789.1 1380.43  4801.1 1371.25  4828.8 1362.11
  4873.4 1358.10  4968.2 1357.32  4978.3 1358.78  4988.2 1353.24  4998.6 1350.30
  5002.6 1345.30  5016.2 1345.30  5017.9 1350.30  5018.1 1351.86  5020.3 1352.00
  5144.4 1354.70  5354.5 1355.14  5401.1 1358.41  5435.1 1358.71  5499.5 1362.82
  5689.5 1365.29  5706.1 1363.25  5712.7 1364.51  5791.6 1366.86  5822.8 1370.61
  5849.4 1375.65  5866.5 1386.75  5893.5 1401.16  5911.3 1408.37  5935.6 1414.48
#Mann=3,-1,0
  4766.2    0.14       0  4998.6    0.04       0  5017.9    0.08       0
#XS Ineff=2,0
       0                 5143.80    0.00 1357.90
Permanent Ineff=
       F       F
Bank Sta=4998.6,5017.9
XS Rating Curve= 0
Exp/Cntr=0.3,0.1

Type RM Length L Ch R = 1,212999,482,482,482
BEGIN DESCRIPTION:
Fisher River 426.0
END DESCRIPTION:
XS GIS Cut Line= 4
      1452422.37      1017715.51      1452245.36      1017373.29
      1452316.17      1017137.28      1452000.51      1016780.32
#Sta/Elev= 30
  4448.4 1383.48  4466.7 1377.82  4480.2 1376.12  4522.2 1361.56  4561.2 1358.97
  4597.7 1359.10  4617.5 1356.13  4720.0 1355.60  4730.7 1354.62  4740.3 1355.43
  4781.1 1355.09  4899.4 1351.87  4918.2 1350.22  4955.1 1350.81  4974.2 1347.02
  4992.0 1345.80  4994.5 1340.30  5005.5 1340.30  5008.0 1345.80  5040.7 1347.93
  5058.1 1352.63  5299.0 1353.84  5307.8 1353.61  5325.9 1350.76  5335.3 1353.21
  5342.5 1357.37  5371.1 1361.52  5406.1 1369.41  5516.1 1382.91  5556.6 1386.70
#Mann=3,-1,0
  4448.4    0.14       0  4992.0    0.04       0  5008.0    0.08       0
#XS Ineff=2,0
       0                 5105.40    0.00 1353.79
Permanent Ineff=
       F       F
Bank Sta=4992,5008
XS Rating Curve= 0
Exp/Cntr=0.3,0.1

Type RM Length L Ch R = 1,212517,501,501,501
BEGIN DESCRIPTION:
Fisher River 425.0
END DESCRIPTION:
XS GIS Cut Line= 3
      1452746.92      1017090.11      1452513.83      1016895.37
      1452074.22      1016685.90
#Sta/Elev= 30
  4797.1 1401.66  4831.7 1390.10  4849.7 1383.44  4864.9 1376.48  4870.5 1373.31
  4899.6 1352.84  4923.8 1346.44  4954.1 1344.30  4962.9 1345.40  4975.5 1346.21
  4990.9 1341.45  4993.4 1336.45  5006.6 1336.45  5009.1 1341.45  5045.5 1349.66
  5052.4 1349.15  5062.5 1349.60  5141.8 1348.29  5199.7 1348.45  5215.2 1349.04
  5232.5 1348.79  5292.1 1349.70  5386.5 1353.06  5416.3 1356.12  5457.9 1364.55
  5467.5 1365.61  5496.8 1366.95  5524.9 1369.48  5548.9 1372.72  5587.8 1376.48
#Mann=3,-1,0
  4797.1    0.14       0  4990.9    0.04       0  5009.1    0.08       0
Bank Sta=4990.9,5009.1
XS Rating Curve= 0
Exp/Cntr=0.3,0.1

Type RM Length L Ch R = 1,212016,529,529,529
BEGIN DESCRIPTION:
Fisher River 424.0
END DESCRIPTION:
XS GIS Cut Line= 3
      1453139.23      1016880.58      1453050.75      1016765.57
      1452266.04      1016004.45
#Sta/Elev= 30
  4801.3 1426.22  4823.5 1416.65  4837.4 1406.32  4852.3 1398.03  4906.8 1356.59
  4915.4 1351.22  4926.2 1346.73  4934.5 1345.38  4949.9 1344.25  4976.4 1339.71
  4990.9 1339.37  4993.4 1333.37  5006.6 1333.37  5009.1 1339.37  5031.2 1341.45
  5095.2 1343.61  5150.9 1343.56  5239.7 1346.02  5441.4 1343.80  5603.7 1344.56
  5647.3 1346.03  5685.2 1344.79  5688.1 1345.25  5715.7 1357.14  5740.8 1361.78
  5771.3 1365.10  5823.3 1368.04  5935.3 1371.55  6006.4 1375.20  6039.6 1378.42
#Mann=3,-1,0
  4801.3    0.14       0  4990.9    0.04       0  5009.1    0.08       0
#XS Ineff=2,0
       0                 5239.70    0.00 1346.02
Permanent Ineff=
       F       F
Bank Sta=4990.9,5009.1
XS Rating Curve= 0
Exp/Cntr=0.3,0.1

Type RM Length L Ch R = 1,211487,500,500,500
BEGIN DESCRIPTION:
Fisher River 423.0
END DESCRIPTION:
XS GIS Cut Line= 4
      1453339.85      1016314.19      1453233.66      1016278.79
      1453003.55      1016293.54      1452322.03      1015939.51
#Sta/Elev= 30
  4847.0 1393.33  4888.8 1376.01  4894.1 1374.52  4953.3 1343.44  4977.5 1337.38
  4990.9 1335.05  4993.4 1328.05  5006.6 1328.05  5009.1 1335.05  5028.6 1339.00
  5044.6 1338.26  5073.8 1339.33  5129.7 1338.39  5197.9 1338.97  5289.3 1341.95
  5319.3 1342.24  5382.8 1341.48  5417.8 1339.50  5436.8 1341.12  5537.4 1342.88
  5613.6 1342.71  5639.6 1340.57  5644.8 1342.32  5677.7 1357.25  5689.4 1358.06
  5705.3 1360.77  5745.5 1363.80  5861.9 1368.28  5881.4 1369.95  5957.5 1380.31
#Mann=3,-1,0
  4847.0    0.14       0  4990.9    0.04       0  5009.1    0.08       0
Bank Sta=4990.9,5009.1
XS Rating Curve= 0
Exp/Cntr=0.3,0.1

Type RM Length L Ch R = 1,210987,542,542,542
BEGIN DESCRIPTION:
Fisher River 422.0
END DESCRIPTION:
XS GIS Cut Line= 4
      1453446.06      1016087.02      1453254.31      1015836.27
      1453167.04      1015781.71      1452516.82      1015379.03
#Sta/Elev= 30
  4633.1 1368.16  4691.3 1355.55  4703.2 1354.44  4740.9 1348.14  4775.5 1340.51
  4798.1 1338.43  4834.9 1337.01  4942.2 1335.30  4973.1 1333.50  4990.9 1330.34
  4993.4 1325.34  5006.6 1325.34  5009.1 1330.34  5013.0 1332.43  5030.3 1334.89
  5081.8 1333.47  5114.6 1334.47  5169.6 1333.26  5300.3 1333.99  5425.1 1339.36
  5437.1 1338.33  5456.7 1333.24  5479.3 1339.25  5502.7 1347.20  5518.9 1354.15
  5548.5 1358.09  5586.9 1360.30  5680.3 1362.71  5753.0 1366.29  5816.5 1367.96
#Mann=3,-1,0
  4633.1    0.14       0  4990.9    0.04       0  5009.1    0.08       0
#XS Ineff=2,0
       0                 5424.30    0.00 1339.32
Permanent Ineff=
       F       F
Bank Sta=4990.9,5009.1
XS Rating Curve= 0
Exp/Cntr=0.5,0.3

Type RM Length L Ch R = 1,210445,130,130,130
BEGIN DESCRIPTION:
Old Lowgap Rd - US
END DESCRIPTION:
XS GIS Cut Line= 6
      1454050.88      1015393.76      1453814.83      1015370.36
      1453469.67      1015379.00      1452850.14      1015364.25
      1452735.09      1015358.35      1452507.91      1015328.85
#Sta/Elev= 30
  4056.9 1369.32  4080.1 1367.35  4115.2 1357.80  4153.2 1351.31  4164.7 1351.80
  4170.2 1349.13  4182.8 1348.75  4226.9 1342.56  4249.7 1342.04  4256.4 1343.13
  4271.3 1340.26  4314.7 1339.41  4326.3 1336.87  4413.0 1340.09  4670.0 1334.12
  4831.7 1332.67  4905.1 1328.91  4977.5 1328.90  4983.7 1322.10  5020.3 1322.10
  5023.9 1328.90  5040.6 1331.96  5047.4 1330.49  5073.3 1331.16  5129.5 1333.16
  5157.3 1335.58  5188.8 1340.62  5214.7 1350.23  5274.9 1359.35  5603.4 1369.55
#Mann=3,-1,0
  4056.9    0.14       0  4977.5    0.04       0  5023.9    0.08       0
#XS Ineff=2,0
    0.00 4966.00 1334.70 5034.00    0.00 1335.17
Permanent Ineff=
       F       F
Bank Sta=4977.5,5023.9
XS Rating Curve= 0
Exp/Cntr=0.5,0.3

Type RM Length L Ch R =3,210375,,,
BEGIN DESCRIPTION:
Old Lowgap Rd - TOR
Structure ID: LDS_FR_23
Approximate Survey Structure
END DESCRIPTION:
Bridge Culvert--1,0,-1,-1,0
Deck Dist Width WeirC Skew NumUp NumDn MinLoCord MaxHiCord MaxSubmerge Is_Ogee
55,30,3,,37,37,,,0.95,0,1,1,,,
  4165.6  4180.3  4274.7  4365.2  4430.4  4449.6  4471.6  4474.3  4528.2  4579.4
  4590.3  4600.0  4622.5  4682.3  4682.8  4710.2  4768.2  4976.0  4976.0  5024.0
  5024.0  5098.5  5112.7  5133.8  5139.8  5174.1  5200.5  5239.8  5245.4  5257.7
  5266.3  5302.1  5325.2  5331.9  5334.0  5346.8  5353.5
 1349.46 1348.85 1345.70 1343.14 1341.70 1341.31 1340.80 1340.69 1339.32 1337.92
 1337.67 1337.44 1336.82 1335.69 1335.67 1335.22 1334.76 1334.70 1334.70 1334.70
 1334.70 1337.69 1338.24 1339.36 1339.65 1341.46 1343.11 1345.93 1346.23 1347.12
 1347.67 1349.81 1351.42 1351.56 1351.65 1352.43 1352.73
 1302.10 1302.10 1302.10 1302.10 1302.10 1302.10 1302.10 1302.10 1302.10 1302.10
 1302.10 1302.10 1302.10 1302.10 1302.10 1302.10 1302.10 1302.10 1332.70 1332.70
 1302.10 1302.10 1302.10 1302.10 1302.10 1302.10 1302.10 1302.10 1302.10 1302.10
 1302.10 1302.10 1302.10 1302.10 1302.10 1302.10 1302.10
  4165.6  4180.3  4274.7  4365.2  4430.4  4449.6  4471.6  4474.3  4528.2  4579.4
  4590.3  4600.0  4622.5  4682.3  4682.8  4710.2  4768.2  4976.0  4976.0  5024.0
  5024.0  5098.5  5112.7  5133.8  5139.8  5174.1  5200.5  5239.8  5245.4  5257.7
  5266.3  5302.1  5325.2  5331.9  5334.0  5346.8  5353.5
 1349.46 1348.85 1345.70 1343.14 1341.70 1341.31 1340.80 1340.69 1339.32 1337.92
 1337.67 1337.44 1336.82 1335.69 1335.67 1335.22 1334.76 1334.70 1334.70 1334.70
 1334.70 1337.69 1338.24 1339.36 1339.65 1341.46 1343.11 1345.93 1346.23 1347.12
 1347.67 1349.81 1351.42 1351.56 1351.65 1352.43 1352.73
 1302.10 1302.10 1302.10 1302.10 1302.10 1302.10 1302.10 1302.10 1302.10 1302.10
 1302.10 1302.10 1302.10 1302.10 1302.10 1302.10 1302.10 1302.10 1332.70 1332.70
 1302.10 1302.10 1302.10 1302.10 1302.10 1302.10 1302.10 1302.10 1302.10 1302.10
 1302.10 1302.10 1302.10 1302.10 1302.10 1302.10 1302.10
BR Coef=1,1,0,1.25,0,,,0.8,0,2,0,
WSPro=,,,, 1 ,,,, 0 ,,,, 0 ,,,,-1 ,-1 ,-1 , 0 , 0 , 0 , 0 , 0
BC Design=,,0,,0,,,,,,

Type RM Length L Ch R = 1,210315,315,315,315
BEGIN DESCRIPTION:
Old Lowgap Rd - DS
END DESCRIPTION:
XS GIS Cut Line= 5
      1453717.45      1015119.41      1453469.67      1015252.15
      1453062.55      1015240.35      1452847.19      1015228.55
      1452661.30      1015089.86
#Sta/Elev= 30
  4371.9 1371.09  4390.0 1367.36  4452.3 1338.22  4490.3 1333.21  4492.0 1331.21
  4495.8 1330.88  4497.5 1329.72  4505.6 1334.23  4560.6 1332.49  4605.3 1333.40
  4637.7 1332.27  4676.7 1332.93  4780.5 1330.09  4862.3 1331.09  4910.6 1330.40
  4927.5 1331.68  4945.8 1331.20  4961.1 1328.34  4977.5 1327.65  4986.5 1321.85
  5013.5 1321.85  5022.5 1327.65  5024.9 1328.97  5140.1 1333.16  5261.5 1341.53
  5305.5 1346.99  5365.6 1359.05  5392.2 1362.19  5447.0 1365.95  5507.9 1368.64
#Mann=5,-1,0
  4371.9    0.08       0  4605.3    0.14       0  4977.5    0.04       0
  5022.5    0.08       0  5261.5    0.14       0
#XS Ineff=2,0
    0.00 4966.00 1334.00 5034.00    0.00 1334.00
Permanent Ineff=
       F       F
Bank Sta=4977.5,5022.5
XS Rating Curve= 0
Exp/Cntr=0.5,0.3

Type RM Length L Ch R = 1,210000,495,495,495
BEGIN DESCRIPTION:
Fisher River 420.0
END DESCRIPTION:
XS GIS Cut Line= 5
      1453720.42      1015016.14      1453292.66      1015019.09
      1453101.53      1014929.22      1452954.93      1014863.65
      1452850.14      1014845.03
#Sta/Elev= 30
  4396.2 1376.18  4434.7 1368.66  4505.0 1347.39  4525.2 1344.09  4537.6 1337.83
  4576.4 1333.16  4592.7 1327.25  4615.9 1327.72  4630.5 1324.58  4635.8 1331.56
  4665.8 1329.48  4707.1 1330.20  4731.2 1326.27  4760.1 1324.51  4915.3 1326.52
  4970.9 1323.62  4990.9 1323.62  4993.4 1318.62  5006.6 1318.62  5009.1 1323.62
  5011.9 1325.20  5036.8 1328.40  5082.4 1328.35  5137.3 1330.16  5155.4 1335.66
  5162.7 1336.42  5181.7 1344.40  5200.9 1348.12  5242.3 1353.25  5302.2 1357.59
#Mann=5,-1,0
  4396.2    0.14       0  4990.9    0.04       0  5009.1    0.14       0
  5082.4    0.08       0  5200.9    0.14       0
#XS Ineff=2,0
    0.00 4707.10 1330.10               0
Permanent Ineff=
       F       F
Bank Sta=4990.9,5009.1
XS Rating Curve= 0
Exp/Cntr=0.3,0.1

Type RM Length L Ch R = 1,209505,496,496,496
BEGIN DESCRIPTION:
Fisher River 419.0
END DESCRIPTION:
XS GIS Cut Line= 4
      1453773.55      1014624.36      1453422.47      1014633.21
      1453257.26      1014630.26      1452859.01      1014774.81
#Sta/Elev= 30
  4580.1 1363.95  4636.1 1346.30  4678.1 1339.18  4691.9 1337.66  4718.3 1333.77
  4796.4 1325.85  4813.7 1324.71  4884.9 1322.72  4938.1 1323.20  4959.3 1323.07
  4990.9 1317.67  4993.4 1312.67  5010.1 1312.67  5013.3 1317.67  5015.1 1317.67
  5030.5 1322.09  5047.4 1322.84  5063.1 1325.11  5083.8 1325.18  5131.8 1326.10
  5205.2 1326.55  5238.7 1327.95  5256.7 1329.42  5293.9 1333.97  5309.8 1334.79
  5345.8 1340.56  5369.2 1344.84  5383.5 1346.68  5412.6 1348.33  5520.2 1356.62
#Mann=5,-1,0
  4580.1    0.08       0  4938.1    0.14       0  4990.9    0.04       0
  5013.3    0.14       0  5083.8    0.08       0
Bank Sta=4990.9,5013.3
XS Rating Curve= 0
Exp/Cntr=0.3,0.1

Type RM Length L Ch R = 1,209009,505,505,505
BEGIN DESCRIPTION:
Fisher River 418.0
END DESCRIPTION:
XS GIS Cut Line= 3
      1453755.82      1014205.44      1453328.06      1014187.74
      1452835.40      1014459.15
#Sta/Elev= 30
  4685.2 1373.95  4690.8 1371.50  4715.0 1362.73  4720.4 1360.19  4784.3 1335.07
  4806.1 1328.83  4827.0 1323.62  4851.2 1320.12  4862.5 1319.36  4964.7 1319.10
  4984.6 1317.23  4985.8 1315.88  4989.5 1310.88  5010.5 1310.88  5014.3 1315.88
  5038.5 1318.80  5063.5 1319.84  5251.9 1323.68  5284.8 1325.02  5328.8 1325.92
  5370.0 1328.08  5421.7 1329.02  5497.0 1330.60  5537.5 1334.07  5551.7 1334.40
  5569.5 1338.58  5610.0 1351.46  5643.0 1365.05  5651.3 1367.04  5675.8 1369.59
#Mann=4,-1,0
  4685.2    0.14       0  4985.8    0.04       0  5014.3    0.08       0
  5421.7    0.14       0
Bank Sta=4985.8,5014.3
XS Rating Curve= 0
Exp/Cntr=0.3,0.1

Type RM Length L Ch R = 1,208504,496,496,496
BEGIN DESCRIPTION:
Fisher River 417.0
END DESCRIPTION:
XS GIS Cut Line= 3
      1453502.12      1013657.31      1453286.76      1013793.01
      1452879.61      1013925.78
#Sta/Elev= 30
  4858.2 1372.62  4877.1 1368.28  4905.8 1354.78  4914.7 1351.94  4927.4 1345.13
  4942.5 1342.05  4948.4 1337.52  4964.3 1323.01  4986.2 1314.92  4989.6 1310.80
  4990.5 1310.80  4993.0 1305.80  5007.0 1305.80  5009.5 1310.80  5026.6 1314.22
  5045.1 1315.92  5060.4 1313.98  5135.6 1317.09  5156.9 1316.36  5275.3 1317.73
  5357.2 1316.70  5377.7 1319.87  5399.0 1322.08  5415.6 1328.31  5439.5 1340.64
  5471.7 1353.22  5498.7 1359.54  5512.3 1361.66  5526.6 1362.28  5541.0 1364.92
#Mann=4,-1,0
  4858.2    0.14       0  4990.5    0.04       0  5009.5    0.08       0
  5275.3    0.14       0
#XS Ineff=2,0
       0                 5285.00    0.00 1317.89
Permanent Ineff=
       F       F
Bank Sta=4990.5,5009.5
XS Rating Curve= 0
Exp/Cntr=0.3,0.1

Type RM Length L Ch R = 1,208008,515,515,515
BEGIN DESCRIPTION:
Fisher River 416.0
END DESCRIPTION:
XS GIS Cut Line= 3
      1453413.64      1013350.49      1453056.65      1013344.59
      1452820.66      1013477.34
#Sta/Elev= 30
  4732.4 1367.77  4765.7 1359.87  4776.3 1356.91  4812.8 1341.25  4865.0 1317.79
  4868.2 1316.87  4873.2 1315.75  4906.3 1313.32  4953.4 1312.87  4975.0 1311.22
  4990.5 1305.69  4993.0 1300.69  5007.0 1300.69  5009.5 1305.69  5024.4 1312.37
  5062.2 1312.68  5096.5 1314.08  5107.8 1314.89  5119.3 1315.30  5131.8 1316.05
  5156.7 1318.54  5205.2 1325.22  5217.2 1327.27  5228.0 1330.35  5263.0 1339.72
  5266.7 1341.06  5285.4 1346.90  5327.3 1358.79  5336.3 1360.69  5360.2 1363.88
#Mann=4,-1,0
  4732.4    0.14       0  4990.5    0.04       0  5009.5    0.08       0
  5228.0    0.14       0
Bank Sta=4990.5,5009.5
XS Rating Curve= 0
Exp/Cntr=0.3,0.1

Type RM Length L Ch R = 1,207493,493,493,493
BEGIN DESCRIPTION:
Fisher River 415.0
END DESCRIPTION:
XS GIS Cut Line= 4
      1453693.85      1013121.84      1453413.62      1012930.10
      1453319.21      1012865.20      1453215.95      1012708.83
#Sta/Elev= 30
  4588.1 1371.58  4593.0 1369.33  4611.5 1362.80  4618.1 1358.69  4632.0 1351.36
  4658.6 1335.48  4688.7 1321.15  4698.3 1317.40  4712.7 1314.84  4778.2 1309.84
  4817.7 1308.83  4934.0 1308.73  4960.2 1308.27  4973.7 1306.45  4980.1 1304.27
  4990.5 1301.93  4993.0 1296.93  5007.0 1296.93  5009.5 1301.93  5013.5 1305.26
  5056.7 1306.89  5069.8 1314.30  5104.8 1336.01  5116.7 1345.38  5133.5 1353.16
  5151.8 1359.22  5179.6 1362.73  5208.8 1364.37  5222.4 1365.94  5229.6 1365.89
#Mann=5,-1,0
  4588.1    0.14       0  4688.7    0.08       0  4934.0    0.14       0
  4990.5    0.04       0  5009.5    0.14       0
Bank Sta=4990.5,5009.5
XS Rating Curve= 0
Exp/Cntr=0.3,0.1

Type RM Length L Ch R = 1,207000,507,507,507
BEGIN DESCRIPTION:
Fisher River 414.0
END DESCRIPTION:
XS GIS Cut Line= 3
      1453925.00      1012875.00      1453597.36      1012476.24
      1453174.96      1012274.98
#Sta/Elev= 30
  4483.9 1331.37  4510.3 1324.82  4550.7 1318.25  4668.1 1307.45  4766.4 1304.02
  4877.3 1303.33  4919.9 1304.34  4948.0 1302.90  4962.5 1303.67  4976.2 1301.07
  4982.6 1298.12  4984.3 1293.12  5007.0 1293.12  5009.5 1298.12  5012.5 1302.09
  5018.5 1303.52  5070.2 1302.59  5113.3 1305.98  5200.2 1309.41  5245.3 1312.38
  5261.8 1315.05  5305.5 1324.30  5332.6 1333.47  5335.3 1336.13  5340.8 1335.91
  5362.8 1342.35  5382.9 1346.81  5414.7 1352.85  5438.8 1355.84  5467.9 1358.05
#Mann=3,-1,0
  4483.9    0.08       0  4982.6    0.04       0  5009.5    0.08       0
Bank Sta=4982.6,5009.5
XS Rating Curve= 0
Exp/Cntr=0.3,0.1

Type RM Length L Ch R = 1,206493,490,490,490
BEGIN DESCRIPTION:
Fisher River 413.0
END DESCRIPTION:
XS GIS Cut Line= 4
      1454508.13      1012248.62      1453968.24      1012118.81
      1453835.48      1012118.81      1453384.07      1011983.10
#Sta/Elev= 30
  4373.5 1333.50  4396.0 1333.28  4457.0 1325.49  4528.6 1312.52  4541.5 1312.38
  4595.7 1308.04  4644.0 1305.35  4774.9 1300.36  4809.5 1301.25  4925.3 1300.99
  4958.9 1302.01  4990.5 1293.80  4993.0 1288.80  5007.0 1288.80  5009.5 1293.80
  5011.7 1295.95  5028.4 1297.73  5119.4 1297.28  5217.8 1299.50  5313.7 1299.60
  5357.9 1300.46  5388.9 1302.64  5409.4 1308.22  5419.4 1312.27  5444.2 1319.40
  5473.1 1323.32  5482.4 1329.68  5491.1 1333.14  5520.1 1341.29  5532.9 1343.99
#Mann=3,-1,0
  4373.5    0.08       0  4990.5    0.04       0  5009.5    0.08       0
Bank Sta=4990.5,5009.5
XS Rating Curve= 0
Exp/Cntr=0.3,0.1

Type RM Length L Ch R = 1,206003,503,503,503
BEGIN DESCRIPTION:
Fisher River 412.0
END DESCRIPTION:
XS GIS Cut Line= 3
      1454561.20      1012036.20      1453956.44      1011605.49
      1453625.04      1011525.01
#Sta/Elev= 30
  4411.4 1322.94  4473.3 1319.00  4535.5 1312.75  4617.6 1307.97  4701.2 1304.67
  4788.1 1299.83  4906.4 1297.22  4950.7 1294.80  4957.5 1293.79  4964.2 1294.11
  4975.4 1292.90  4990.5 1288.80  4993.0 1283.80  5007.0 1283.80  5009.5 1288.80
  5013.1 1288.83  5027.8 1292.40  5102.0 1291.18  5148.2 1292.11  5174.7 1290.22
  5191.3 1290.41  5219.3 1291.86  5249.6 1296.51  5278.0 1302.69  5307.6 1311.51
  5359.8 1329.69  5382.7 1335.72  5398.7 1338.23  5423.2 1340.78  5494.9 1346.32
#Mann=3,-1,0
  4411.4    0.08       0  4990.5    0.04       0  5009.5    0.08       0
Bank Sta=4990.5,5009.5
XS Rating Curve= 0
Exp/Cntr=0.3,0.1

Type RM Length L Ch R = 1,205500,506,506,506
BEGIN DESCRIPTION:
Fisher River 411.0
END DESCRIPTION:
XS GIS Cut Line= 4
      1454581.88      1011248.53      1454278.00      1011233.78
      1454177.70      1011204.27      1453587.66      1011325.23
#Sta/Elev= 30
  4643.2 1346.81  4669.8 1338.27  4685.8 1329.81  4737.6 1305.89  4755.4 1303.56
  4772.6 1302.16  4868.7 1295.46  4911.9 1290.75  4984.7 1288.70  4990.5 1284.18
  4993.0 1279.18  5007.0 1279.18  5009.5 1284.18  5010.2 1287.33  5019.9 1288.49
  5037.1 1287.52  5118.3 1290.75  5145.0 1290.34  5238.4 1291.77  5272.7 1291.55
  5319.4 1293.90  5361.5 1293.79  5417.8 1295.65  5461.1 1297.90  5488.7 1300.22
  5501.7 1300.52  5536.9 1306.03  5562.1 1311.13  5596.9 1320.92  5654.3 1340.33
#Mann=4,-1,0
  4643.2    0.14       0  4737.6    0.08       0  4990.5    0.04       0
  5009.5    0.08       0
Bank Sta=4990.5,5009.5
XS Rating Curve= 0
Exp/Cntr=0.3,0.1

Type RM Length L Ch R = 1,204994,400,400,400
BEGIN DESCRIPTION:
Fisher River 410.0
END DESCRIPTION:
XS GIS Cut Line= 3
      1454525.03      1010925.02      1454316.36      1010749.36
      1453667.28      1010646.10
#Sta/Elev= 30
  4787.4 1333.72  4820.8 1323.11  4847.5 1313.08  4867.1 1303.41  4902.0 1296.13
  4925.6 1292.68  4956.2 1290.01  4973.7 1284.45  4983.9 1279.34  4990.5 1278.29
  4993.0 1273.29  5007.0 1273.29  5009.5 1278.29  5012.4 1280.34  5018.8 1281.80
  5027.3 1287.01  5098.3 1285.89  5213.7 1287.08  5256.6 1286.60  5531.5 1289.84
  5562.1 1291.33  5592.7 1294.82  5605.0 1301.83  5611.2 1304.05  5615.2 1307.92
  5623.1 1310.58  5630.8 1317.99  5666.0 1329.15  5680.7 1332.55  5717.4 1334.64
#Mann=3,-1,0
  4787.4    0.08       0  4990.5    0.04       0  5009.5    0.08       0
Bank Sta=4990.5,5009.5
XS Rating Curve= 0
Exp/Cntr=0.5,0.3

Type RM Length L Ch R = 1,204594,42,42,42
BEGIN DESCRIPTION:
Off Highway 89 - US
END DESCRIPTION:
XS GIS Cut Line= 3
      1454885.77      1010598.93      1454275.05      1010306.84
      1453693.91      1010504.49
#Sta/Elev= 30
  4645.2 1332.13  4682.3 1320.63  4711.7 1313.22  4721.1 1309.89  4731.4 1309.02
  4754.3 1304.66  4778.8 1301.23  4815.6 1298.57  4841.8 1295.16  4891.5 1284.14
  4948.4 1281.05  4964.4 1281.23  4980.2 1278.03  4984.0 1275.70  4991.6 1269.90
  5008.4 1269.90  5016.0 1275.70  5026.7 1280.10  5069.5 1283.98  5298.7 1283.07
  5472.2 1285.99  5593.0 1286.55  5657.4 1288.26  5757.3 1287.78  5797.9 1288.67
  5810.7 1289.90  5851.5 1296.97  5897.7 1316.74  5921.4 1323.72  5936.0 1324.84
#Mann=3,-1,0
  4645.2    0.08       0  4984.0    0.04       0  5016.0    0.08       0
#XS Ineff=2,0
    0.00 4970.00 1283.20 5030.00    0.00 1283.20
Permanent Ineff=
       F       F
Bank Sta=4984,5016
XS Rating Curve= 0
Exp/Cntr=0.5,0.3

Type RM Length L Ch R =3,204570,,,
BEGIN DESCRIPTION:
Off Highway 89 - TOR
Structure ID: LDS_FR_21
Approximate Survey Structure
END DESCRIPTION:
Bridge Culvert--1,0,-1,-1,0
Deck Dist Width WeirC Skew NumUp NumDn MinLoCord MaxHiCord MaxSubmerge Is_Ogee
18,12,3,,11,11,,,0.95,0,1,1,,,
  4884.7  4899.9  4918.6  4941.7  4966.1  4980.0  4980.0  5020.0  5020.0  5032.2
  5114.9
 1286.75 1285.34 1284.13 1283.57 1283.20 1283.20 1283.20 1283.20 1283.20 1283.20
 1283.40
 1249.90 1249.90 1249.90 1249.90 1249.90 1249.90 1281.20 1281.20 1249.90 1249.90
 1249.90
  4884.7  4899.9  4918.6  4941.7  4966.1  4980.0  4980.0  5020.0  5020.0  5032.2
  5114.9
 1286.75 1285.34 1284.13 1283.57 1283.20 1283.20 1283.20 1283.20 1283.20 1283.20
 1283.40
 1249.90 1249.90 1249.90 1249.90 1249.90 1249.90 1281.20 1281.20 1249.90 1249.90
 1249.90
BR Coef=1,1,0,1.25,0,,,0.8,0,2,0,
WSPro=,,,, 1 ,,,, 0 ,,,, 0 ,,,,-1 ,-1 ,-1 , 0 , 0 , 0 , 0 , 0
BC Design=,,0,,0,,,,,,

Type RM Length L Ch R = 1,204552,623,623,623
BEGIN DESCRIPTION:
Off Highway 89 - DS
END DESCRIPTION:
XS GIS Cut Line= 3
      1454909.35      1010560.56      1454263.25      1010256.69
      1453685.01      1010463.21
#Sta/Elev= 30
  4644.8 1333.59  4669.6 1325.17  4706.7 1313.85  4749.0 1304.62  4778.2 1299.96
  4816.9 1297.12  4843.5 1294.06  4896.9 1284.80  4922.9 1282.95  4957.0 1283.21
  4968.3 1282.52  4984.0 1276.45  4991.6 1269.65  5008.4 1269.65  5016.0 1276.45
  5026.3 1281.14  5084.8 1283.51  5318.8 1282.74  5465.9 1285.31  5619.5 1285.68
  5772.8 1287.96  5787.4 1287.22  5813.6 1288.31  5836.2 1289.54  5876.3 1294.38
  5890.6 1298.49  5903.9 1304.13  5931.1 1314.06  5945.2 1318.37  5972.8 1324.10
#Mann=3,-1,0
  4644.8    0.08       0  4984.0    0.04       0  5016.0    0.08       0
#XS Ineff=2,0
    0.00 4970.00 1283.00 5030.00    0.00 1283.00
Permanent Ineff=
       F       F
Bank Sta=4984,5016
XS Rating Curve= 0
Exp/Cntr=0.5,0.3

Type RM Length L Ch R = 1,203929,221,221,221
BEGIN DESCRIPTION:
Fisher River 408.0
END DESCRIPTION:
XS GIS Cut Line= 4
      1455155.34      1009844.68      1454735.27      1009802.37
      1454626.12      1009823.02      1453696.50      1010384.30
#Sta/Elev= 30
  4527.9 1328.65  4560.5 1317.96  4605.4 1302.09  4648.5 1294.93  4679.8 1286.31
  4693.4 1283.87  4728.4 1280.15  4795.1 1275.29  4863.3 1274.26  4922.2 1274.18
  4950.9 1274.90  4972.0 1274.42  4986.3 1272.77  4999.5 1265.97  5026.1 1265.97
  5027.7 1272.77  5054.7 1278.54  5070.1 1279.73  5161.3 1278.64  5213.0 1279.64
  5302.8 1279.80  5500.1 1282.74  5746.2 1284.12  5851.6 1286.64  5927.8 1286.64
  5974.4 1287.76  6022.8 1290.55  6063.5 1295.63  6077.1 1298.79  6147.1 1319.17
#Mann=3,-1,0
  4527.9    0.08       0  4986.3    0.04       0  5027.7    0.08       0
#XS Ineff=2,0
    0.00 4883.00 1278.73               0
Permanent Ineff=
       F       F
Bank Sta=4986.3,5027.7
XS Rating Curve= 0
Exp/Cntr=0.5,0.3

Type RM Length L Ch R = 1,203708,139,139,139
BEGIN DESCRIPTION:
W Pine St (HWY 89) - US
END DESCRIPTION:
XS GIS Cut Line= 6
      1455131.77      1009723.60      1454664.47      1009622.12
      1454454.42      1009624.48      1454315.18      1009655.16
      1454039.04      1009780.25      1453805.39      1010028.07
#Sta/Elev= 30
  4430.2 1319.09  4440.2 1314.71  4457.2 1310.20  4477.3 1308.61  4512.3 1294.98
  4549.4 1283.92  4563.9 1282.02  4684.7 1276.33  4705.0 1273.75  4732.5 1272.43
  4787.2 1272.68  4868.2 1270.56  4945.4 1270.99  4965.0 1269.56  4973.4 1265.26
  5026.6 1265.26  5035.0 1269.56  5051.1 1273.21  5112.7 1277.88  5205.4 1278.58
  5222.7 1280.23  5468.5 1284.16  5502.1 1285.83  5521.1 1287.69  5552.8 1293.73
  5574.8 1295.04  5609.7 1300.32  5692.7 1302.27  5775.7 1306.11  5907.8 1317.35
#Mann=3,-1,0
  4430.2    0.08       0  4965.0    0.04       0  5035.0    0.08       0
#XS Ineff=2,0
    0.00 4965.00 1285.30 5035.00    0.00 1285.30
Permanent Ineff=
       F       F
Bank Sta=4965,5035
XS Rating Curve= 0
Exp/Cntr=0.5,0.3

Type RM Length L Ch R =2,203628,,,
BEGIN DESCRIPTION:
W Pine St (HWY 89) - TOR
Structure ID: LDS_FR_20
Approximate Survey Structure
END DESCRIPTION:
Bridge Culvert--1,0,-1,-1,0
Deck Dist Width WeirC Skew NumUp NumDn MinLoCord MaxHiCord MaxSubmerge Is_Ogee
60,40,3,,13,13,,,0.95,0,1,1,,,
  4405.9  4538.4  4635.0  4730.8  4805.7  4907.5  4972.3  5226.8  5326.0  5409.2
  5452.2  5545.0  5614.7
 1311.32 1301.73 1296.15 1291.92 1289.43 1286.23 1285.30 1285.30 1287.17 1289.31
 1290.57 1294.34 1297.44
 1245.26 1245.26 1245.26 1245.26 1245.26 1245.26 1245.26 1245.26 1245.26 1245.26
 1245.26 1245.26 1245.26
  4405.9  4538.4  4635.0  4730.8  4805.7  4907.5  4972.3  5226.8  5326.0  5409.2
  5452.2  5545.0  5614.7
 1311.32 1301.73 1296.15 1291.92 1289.43 1286.23 1285.30 1285.30 1287.17 1289.31
 1290.57 1294.34 1297.44
 1245.06 1245.06 1245.06 1245.06 1245.06 1245.06 1245.06 1245.06 1245.06 1245.06
 1245.06 1245.06 1245.06
Culvert=4,12,40,40,0.013,0.5,1,29,1,1265.4,5000,1265.2,5000,Culvert #1,0,60
Culvert Bottom n=0.013
Culvert Bottom Depth=0
Culvert Depth Blocked=0
BC Design=,,0,,0,,,,,,
