HEC-RAS study Fisher River.prj: Fisher River Limited Detail Study

--- Fisher River.g01 (geometry) --- (continued)

Type RM Length L Ch R = 1,183607,419,419,419
BEGIN DESCRIPTION:
Fisher River 367.0
END DESCRIPTION:
XS GIS Cut Line= 4
      1462026.91       995774.54      1461815.65       995952.12
      1461743.91       996257.00      1461486.87       996565.85
#Sta/Elev= 30
  4670.7 1223.33  4759.0 1213.30  4776.4 1210.11  4792.5 1205.64  4810.8 1199.39
  4829.6 1195.92  4845.5 1194.95  4897.1 1197.05  4931.9 1197.46  4977.1 1196.18
  4988.5 1188.89  4990.2 1183.89  5042.9 1183.89  5048.0 1188.89  5061.5 1196.01
  5086.2 1197.53  5147.0 1196.84  5159.9 1198.25  5174.3 1202.96  5191.0 1206.26
  5214.4 1209.73  5240.5 1212.51  5405.8 1213.94  5488.7 1213.50  5539.2 1215.41
  5555.9 1217.02  5588.8 1222.63  5604.7 1227.49  5636.1 1239.36  5661.7 1250.60
#Mann=4,-1,0
  4670.7    0.08       0  4829.6    0.14       0  4988.5    0.04       0
  5048.0    0.08       0
Bank Sta=4988.5,5048
XS Rating Curve= 0
Exp/Cntr=0.3,0.1

Type RM Length L Ch R = 1,183188,182,182,182
BEGIN DESCRIPTION:
Fisher River 366.5
END DESCRIPTION:
XS GIS Cut Line= 4
      1461704.06       995589.44      1461450.99       996057.73
      1461383.24       996141.42      1461213.85       996428.38
#Sta/Elev= 30
  4416.4 1246.88  4439.5 1240.29  4495.3 1220.61  4551.6 1214.41  4568.6 1211.61
  4585.1 1207.08  4601.8 1199.70  4623.5 1193.52  4655.2 1193.65  4739.1 1196.75
  4845.2 1196.83  4886.6 1194.88  4932.8 1195.87  4957.5 1196.10  4969.3 1191.94
  4975.1 1188.42  4978.0 1188.42  4980.5 1183.42  5019.5 1183.42  5022.0 1188.42
  5024.6 1192.88  5040.4 1196.07  5085.3 1197.82  5208.4 1203.41  5273.3 1210.39
  5310.6 1216.12  5326.7 1222.55  5347.1 1232.74  5363.0 1238.77  5389.6 1251.38
#Mann=6,-1,0
  4416.4    0.08       0  4932.8    0.14       0  4978.0    0.04       0
  5022.0    0.14       0  5085.3    0.08       0  5347.1    0.14       0
Bank Sta=4978,5022
XS Rating Curve= 0
Exp/Cntr=0.3,0.1

Type RM Length L Ch R = 1,183006,509,509,509
BEGIN DESCRIPTION:
Fisher River 366.0
END DESCRIPTION:
XS GIS Cut Line= 4
      1461690.10       995577.52      1461506.78       995914.26
      1461211.87       995958.10      1460805.35       996217.15
#Sta/Elev= 30
  4470.6 1249.89  4492.2 1242.94  4546.7 1223.58  4558.9 1220.45  4602.6 1215.44
  4640.7 1209.56  4657.9 1200.11  4675.3 1195.62  4691.9 1193.78  4708.4 1193.27
  4763.0 1195.74  4838.4 1196.71  4934.4 1196.00  4972.5 1190.24  4978.0 1187.47
  4980.5 1182.47  5019.5 1182.47  5022.0 1187.47  5031.1 1192.32  5034.9 1193.43
  5072.8 1193.14  5115.4 1197.12  5151.0 1199.16  5167.3 1198.74  5311.5 1207.59
  5416.1 1212.77  5461.5 1216.07  5553.8 1225.30  5568.1 1225.91  5634.2 1238.73
#Mann=5,-1,0
  4470.6    0.08       0  4838.4    0.14       0  4978.0    0.04       0
  5022.0    0.14       0  5167.3    0.08       0
Bank Sta=4978,5022
XS Rating Curve= 0
Exp/Cntr=0.3,0.1

Type RM Length L Ch R = 1,182497,514,514,514
BEGIN DESCRIPTION:
Fisher River 365.0
END DESCRIPTION:
XS GIS Cut Line= 4
      1461369.30       995400.34      1461134.77       995529.58
      1460982.71       995613.56      1460522.41       996171.50
#Sta/Elev= 30
  4667.7 1234.62  4748.3 1231.41  4777.4 1229.68  4794.0 1224.94  4810.5 1218.50
  4839.1 1204.02  4855.5 1196.77  4895.3 1193.01  4920.9 1193.81  4939.2 1194.20
  4961.4 1191.48  4975.8 1185.58  4978.6 1180.58  5021.5 1180.58  5024.2 1185.58
  5028.8 1191.01  5031.3 1192.86  5047.1 1193.93  5061.3 1200.89  5075.0 1205.53
  5089.0 1207.46  5148.9 1210.43  5217.5 1211.44  5358.2 1211.19  5428.4 1213.45
  5632.4 1225.17  5722.8 1232.29  5737.9 1236.50  5768.1 1241.78  5832.5 1258.39
#Mann=6,-1,0
  4667.7    0.14       0  4748.3    0.08       0  4920.9    0.14       0
  4975.8    0.04       0  5024.2    0.14       0  5148.9    0.08       0
Bank Sta=4975.8,5024.2
XS Rating Curve= 0
Exp/Cntr=0.3,0.1

Type RM Length L Ch R = 1,181983,469,469,469
BEGIN DESCRIPTION:
Fisher River 364.0
END DESCRIPTION:
XS GIS Cut Line= 3
      1461343.41       995197.50      1460855.18       995048.04
      1460358.97       995077.93
#Sta/Elev= 30
  4596.5 1233.96  4770.5 1227.23  4793.8 1222.08  4814.3 1213.80  4827.7 1208.10
  4855.9 1191.73  4911.6 1192.15  4956.5 1192.69  4969.1 1188.83  4976.2 1184.68
  4978.7 1179.68  5024.9 1179.68  5028.3 1184.68  5030.2 1184.68  5031.2 1192.05
  5036.1 1194.92  5048.6 1195.00  5060.5 1191.34  5112.4 1190.93  5252.1 1190.04
  5307.2 1192.66  5337.4 1195.37  5361.7 1200.99  5408.8 1203.00  5431.3 1208.37
  5495.7 1212.36  5517.8 1215.32  5527.6 1218.32  5544.4 1220.20  5604.2 1244.26
#Mann=6,-1,0
  4596.5    0.08       0  4911.6    0.14       0  4976.2    0.04       0
  5028.3    0.14       0  5112.4    0.08       0  5527.6    0.14       0
Bank Sta=4976.2,5028.3
XS Rating Curve= 0
Exp/Cntr=0.3,0.1

Type RM Length L Ch R = 1,181514,490,490,490
BEGIN DESCRIPTION:
Fisher River 363.0
END DESCRIPTION:
XS GIS Cut Line= 4
      1461472.92       994736.19      1461066.40       994528.94
      1460906.99       994698.32      1460303.16       994905.58
#Sta/Elev= 30
  4376.7 1228.59  4467.3 1215.29  4520.0 1210.56  4571.0 1207.43  4583.7 1204.50
  4615.0 1203.92  4759.0 1205.68  4819.0 1203.08  4855.7 1202.57  4907.0 1198.68
  4966.8 1193.26  4976.2 1183.38  4978.7 1178.38  5021.3 1178.38  5023.8 1183.38
  5024.3 1188.01  5025.6 1191.23  5029.6 1194.42  5062.2 1189.17  5114.9 1188.83
  5297.1 1190.56  5358.5 1194.12  5373.8 1197.46  5416.2 1198.56  5541.9 1213.23
  5597.7 1214.80  5615.4 1216.72  5655.6 1223.49  5662.0 1223.59  5704.0 1237.53
#Mann=5,-1,0
  4376.7    0.08       0  4907.0    0.14       0  4976.2    0.04       0
  5023.8    0.14       0  5114.9    0.08       0
Bank Sta=4976.2,5023.8
XS Rating Curve= 0
Exp/Cntr=0.5,0.3

Type RM Length L Ch R = 1,181024,55,55,55
BEGIN DESCRIPTION:
Hidden Valley Rd (2) - US
END DESCRIPTION:
XS GIS Cut Line= 4
      1461480.84       994696.30      1460795.40       994251.96
      1460679.82       994325.69      1460548.32       994331.67
#Sta/Elev= 30
  4099.2 1225.26  4140.9 1218.51  4193.2 1212.61  4273.4 1207.36  4284.2 1205.50
  4411.7 1204.32  4526.8 1204.46  4620.5 1202.34  4642.7 1200.27  4676.3 1192.58
  4720.4 1187.47  4776.0 1187.68  4856.9 1190.54  4896.5 1190.17  4928.7 1193.83
  4957.6 1193.05  4973.5 1188.20  4982.5 1177.60  5017.5 1177.60  5026.5 1188.20
  5036.7 1189.12  5067.8 1187.26  5075.3 1188.71  5083.8 1194.24  5096.0 1197.27
  5102.9 1197.27  5125.3 1200.10  5162.6 1217.32  5180.5 1227.63  5184.8 1231.31
#Mann=3,-1,0
  4099.2    0.08       0  4973.5    0.04       0  5026.5    0.14       0
#XS Ineff=2,0
    0.00 4930.00 1197.40 5070.00    0.00 1197.40
Permanent Ineff=
       F       F
Bank Sta=4973.5,5026.5
XS Rating Curve= 0
Exp/Cntr=0.5,0.3

Type RM Length L Ch R =3,180998,,,
BEGIN DESCRIPTION:
Hidden Valley Rd (2) - TOR
Structure ID: LDS_FR_15
Approximate Survey Structure
END DESCRIPTION:
Bridge Culvert--1,0,-1,-1,0
Deck Dist Width WeirC Skew NumUp NumDn MinLoCord MaxHiCord MaxSubmerge Is_Ogee
17,18,3,,23,23,,,0.95,0,1,1,,,
  4373.0  4391.0  4393.5  4402.6  4410.0  4413.6  4417.1  4422.7  4426.1  4433.7
  4443.6  4454.6  4454.7  4496.1  4536.4  4609.4  4622.8  4632.2  4950.0  4950.0
  5050.0  5050.0  5106.3
 1204.20 1203.99 1203.91 1203.76 1203.53 1203.52 1203.43 1203.48 1203.45 1203.28
 1202.94 1202.63 1202.62 1202.27 1202.04 1198.83 1197.88 1197.40 1197.40 1197.40
 1197.40 1197.40 1197.40
 1157.60 1157.60 1157.60 1157.60 1157.60 1157.60 1157.60 1157.60 1157.60 1157.60
 1157.60 1157.60 1157.60 1157.60 1157.60 1157.60 1157.60 1157.60 1157.60 1194.40
 1194.40 1157.60 1157.60
  4373.0  4391.0  4393.5  4402.6  4410.0  4413.6  4417.1  4422.7  4426.1  4433.7
  4443.6  4454.6  4454.7  4496.1  4536.4  4609.4  4622.8  4632.2  4950.0  4950.0
  5050.0  5050.0  5106.3
 1204.20 1203.99 1203.91 1203.76 1203.53 1203.52 1203.43 1203.48 1203.45 1203.28
 1202.94 1202.63 1202.62 1202.27 1202.04 1198.83 1197.88 1197.40 1197.40 1197.40
 1197.40 1197.40 1197.40
 1157.60 1157.60 1157.60 1157.60 1157.60 1157.60 1157.60 1157.60 1157.60 1157.60
 1157.60 1157.60 1157.60 1157.60 1157.60 1157.60 1157.60 1157.60 1157.60 1194.40
 1194.40 1157.60 1157.60
Pier Skew, UpSta & Num, DnSta & Num=,4975,2,4975,2,0,0,0,0,0
       1       1
 1191.43 1194.40
       1       1
 1191.18 1194.40
Pier Skew, UpSta & Num, DnSta & Num=,5025,2,5025,2,0,0,0,0,0
       1       1
 1191.43 1194.40
       1       1
 1191.18 1194.40
BR Coef=1,1,0,1.25,0,,,0.8,0,2,0,
WSPro=,,,, 1 ,,,, 0 ,,,, 0 ,,,,-1 ,-1 ,-1 , 0 , 0 , 0 , 0 , 0
BC Design=,,0,,0,,,,,,

Type RM Length L Ch R = 1,180969,198,198,198
BEGIN DESCRIPTION:
Hidden Valley Rd (2) - DS
END DESCRIPTION:
XS GIS Cut Line= 4
      1461530.68       994650.49      1460811.34       994168.27
      1460643.95       994287.83      1460540.30       994301.78
#Sta/Elev= 30
  3998.0 1224.35  4083.6 1213.98  4183.5 1205.77  4206.0 1207.51  4279.4 1205.42
  4390.4 1204.16  4444.7 1201.10  4539.5 1201.77  4561.8 1200.48  4583.1 1196.97
  4594.4 1193.47  4627.1 1189.21  4650.3 1188.11  4799.4 1189.09  4810.2 1193.07
  4823.0 1195.81  4868.6 1194.83  4912.0 1194.97  4950.7 1191.43  4962.7 1187.95
  4972.7 1177.35  5022.8 1177.35  5034.8 1187.95  5054.8 1188.82  5073.6 1192.54
  5085.5 1200.05  5099.5 1204.33  5110.5 1210.45  5148.8 1227.75  5174.3 1236.27
#Mann=4,-1,0
  3998.0    0.08       0  4868.6    0.14       0  4962.7    0.04       0
  5034.8    0.14       0
#XS Ineff=2,0
    0.00 4930.00 1196.50 5070.00    0.00 1196.50
Permanent Ineff=
       F       F
Bank Sta=4962.7,5034.8
XS Rating Curve= 0
Exp/Cntr=0.5,0.3

Type RM Length L Ch R = 1,180771,260,260,260
BEGIN DESCRIPTION:
Fisher River 362.0
END DESCRIPTION:
XS GIS Cut Line= 4
      1461702.03       994532.91      1460835.25       994146.35
      1460693.77       994034.76      1460663.87       993970.98
#Sta/Elev= 30
  3918.3 1222.05  3942.3 1221.04  3982.9 1216.47  4123.2 1211.02  4192.0 1209.05
  4342.6 1207.26  4430.6 1204.98  4513.3 1199.93  4561.7 1194.55  4653.8 1188.67
  4785.3 1187.88  4799.0 1188.90  4810.3 1194.31  4824.0 1195.40  4885.9 1194.05
  4926.8 1192.72  4947.6 1190.12  4958.4 1189.67  4976.2 1181.18  4978.7 1176.18
  5022.7 1176.18  5023.8 1181.18  5027.8 1181.26  5039.4 1199.52  5047.3 1213.53
  5073.5 1255.76  5086.0 1263.97  5097.7 1276.89  5107.0 1285.46  5118.0 1292.92
#Mann=4,-1,0
  3918.3    0.08       0  4885.9    0.14       0  4976.2    0.04       0
  5023.8    0.14       0
#XS Ineff=2,0
    0.00 4824.00 1195.40               0
Permanent Ineff=
       F       F
Bank Sta=4976.2,5023.8
XS Rating Curve= 0
Exp/Cntr=0.5,0.3

Type RM Length L Ch R = 1,180511,70,70,70
BEGIN DESCRIPTION:
Hidden Valley Rd - US
END DESCRIPTION:
XS GIS Cut Line= 6
      1461702.05       994520.96      1460901.09       994109.25
      1460926.68       994054.42      1460977.85       993924.65
      1460999.79       993860.68      1460941.26       993822.28
#Sta/Elev= 30
  3937.7 1222.13  4003.5 1217.06  4102.9 1212.15  4197.5 1209.18  4398.2 1206.38
  4486.9 1203.94  4543.6 1199.37  4590.3 1193.55  4670.8 1188.54  4776.3 1187.55
  4789.8 1188.57  4800.7 1193.85  4820.3 1195.37  4852.1 1193.01  4863.5 1193.94
  4892.0 1191.44  4944.6 1190.57  4954.4 1187.30  4969.1 1175.10  5025.8 1175.10
  5032.1 1187.30  5044.3 1189.51  5054.9 1197.10  5086.9 1197.66  5099.0 1199.77
  5105.9 1198.76  5125.4 1207.03  5158.4 1219.46  5163.2 1221.78  5175.9 1231.90
#Mann=4,-1,0
  3937.7    0.08       0  4820.3    0.14       0  4954.4    0.04       0
  5032.1    0.14       0
#XS Ineff=2,0
    0.00 4940.00 1197.70 5060.00    0.00 1197.70
Permanent Ineff=
       F       F
Bank Sta=4954.4,5032.1
XS Rating Curve= 0
Exp/Cntr=0.5,0.3

Type RM Length L Ch R =3,180482,,,
BEGIN DESCRIPTION:
Hidden Valley Rd - TOR
Structure ID: LDS_FR_14
Approximate Survey Structure
END DESCRIPTION:
Bridge Culvert--1,0,-1,-1,0
Deck Dist Width WeirC Skew NumUp NumDn MinLoCord MaxHiCord MaxSubmerge Is_Ogee
35,20,3,,19,19,,,0.95,0,1,1,,,
  4285.7  4367.9  4406.7  4421.4  4465.9  4492.1  4511.4  4522.0  4534.9  4545.0
  4557.7  4564.7  4571.0  4587.1  4950.0  4950.0  5050.0  5050.0  5157.2
 1207.75 1207.11 1206.47 1206.30 1205.17 1204.44 1204.02 1203.45 1202.62 1201.84
 1200.41 1199.52 1198.83 1197.70 1197.70 1197.70 1197.70 1197.70 1197.96
 1155.10 1155.10 1155.10 1155.10 1155.10 1155.10 1155.10 1155.10 1155.10 1155.10
 1155.10 1155.10 1155.10 1155.10 1155.10 1195.20 1195.20 1155.10 1155.10
  4285.7  4367.9  4406.7  4421.4  4465.9  4492.1  4511.4  4522.0  4534.9  4545.0
  4557.7  4564.7  4571.0  4587.1  4950.0  4950.0  5050.0  5050.0  5157.2
 1207.75 1207.11 1206.47 1206.30 1205.17 1204.44 1204.02 1203.45 1202.62 1201.84
 1200.41 1199.52 1198.83 1197.70 1197.70 1197.70 1197.70 1197.70 1197.96
 1155.10 1155.10 1155.10 1155.10 1155.10 1155.10 1155.10 1155.10 1155.10 1155.10
 1155.10 1155.10 1155.10 1155.10 1155.10 1195.20 1195.20 1155.10 1155.10
Pier Skew, UpSta & Num, DnSta & Num=,4975,2,4975,2,0,0,0,0,0
       1       1
 1186.70 1195.20
       1       1
 1186.45 1195.20
Pier Skew, UpSta & Num, DnSta & Num=,5025,2,5025,2,0,0,0,0,0
       1       1
 1186.70 1195.20
       1       1
 1186.45 1195.20
BR Coef=1,1,0,1.25,0,,,0.8,0,2,0,
WSPro=,,,, 1 ,,,, 0 ,,,, 0 ,,,,-1 ,-1 ,-1 , 0 , 0 , 0 , 0 , 0
BC Design=,,0,,0,,,,,,

Type RM Length L Ch R = 1,180441,433,433,433
BEGIN DESCRIPTION:
Hidden Valley Rd - DS
END DESCRIPTION:
XS GIS Cut Line= 6
      1461718.04       994481.14      1460996.66       994110.48
      1461020.57       994028.78      1461042.49       993905.23
      1461054.45       993853.42      1460958.78       993779.68
#Sta/Elev= 30
  4032.0 1221.80  4170.5 1213.79  4272.2 1209.72  4436.6 1207.03  4564.3 1203.28
  4618.2 1199.31  4640.3 1196.32  4662.4 1194.18  4675.6 1193.98  4685.1 1192.49
  4722.5 1191.25  4753.9 1188.65  4831.3 1187.10  4904.2 1186.73  4916.5 1187.76
  4953.5 1187.05  4963.7 1174.85  5020.7 1174.85  5030.9 1187.05  5052.2 1190.71
  5073.9 1191.95  5098.0 1195.84  5138.1 1197.37  5149.0 1195.41  5157.5 1200.40
  5168.4 1208.15  5175.9 1211.82  5187.0 1214.95  5214.3 1234.21  5227.6 1240.33
#Mann=4,-1,0
  4032.0    0.08       0  4831.3    0.14       0  4953.5    0.04       0
  5030.9    0.14       0
#XS Ineff=2,0
    0.00 4940.00 1196.50 5060.00    0.00 1196.50
Permanent Ineff=
       F       F
Bank Sta=4953.5,5030.9
XS Rating Curve= 0
Exp/Cntr=0.5,0.3

Type RM Length L Ch R = 1,180008,512,512,512
BEGIN DESCRIPTION:
Fisher River 360.0
END DESCRIPTION:
XS GIS Cut Line= 4
      1461743.30       994422.20      1461629.01       994358.20
      1461423.33       993818.88      1461098.83       993503.51
#Sta/Elev= 30
  4377.2 1222.12  4486.6 1215.40  4691.2 1205.68  4783.9 1202.31  4849.9 1203.93
  4868.0 1200.90  4905.0 1189.09  4929.7 1187.35  4955.4 1189.40  4960.0 1187.52
  4968.7 1179.48  4971.4 1179.48  4978.7 1174.48  5021.3 1174.48  5028.7 1179.48
  5030.6 1179.48  5030.9 1181.38  5042.9 1187.93  5099.3 1185.58  5189.0 1187.94
  5269.6 1187.23  5320.8 1188.69  5338.1 1191.31  5359.5 1200.10  5390.4 1200.75
  5410.2 1210.63  5452.6 1236.34  5483.0 1257.00  5505.5 1279.50  5537.9 1302.11
#Mann=4,-1,0
  4377.2    0.08       0  4971.4    0.04       0  5028.7    0.08       0
  5410.2    0.14       0
#XS Ineff=2,0
       0                 5042.90    0.00 1191.00
Permanent Ineff=
       F       F
Bank Sta=4971.4,5028.7
XS Rating Curve= 0
Exp/Cntr=0.3,0.1

Type RM Length L Ch R = 1,179496,498,498,498
BEGIN DESCRIPTION:
Fisher River 359.0
END DESCRIPTION:
XS GIS Cut Line= 4
      1462086.08       994344.51      1461960.84       994171.21
      1461939.80       993594.92      1461450.75       992987.02
#Sta/Elev= 30
  4387.0 1237.04  4476.5 1232.49  4560.1 1230.61  4666.8 1216.62  4710.6 1207.57
  4748.7 1194.34  4775.7 1187.57  4856.3 1184.81  4899.5 1185.96  4962.1 1186.42
  4965.9 1184.58  4969.1 1179.26  4971.8 1174.26  5021.3 1174.26  5025.2 1179.26
  5026.6 1179.26  5028.3 1182.59  5029.0 1189.50  5035.7 1187.39  5266.2 1183.77
  5397.6 1185.82  5488.1 1189.91  5682.5 1187.74  5728.2 1189.43  5740.6 1192.09
  5784.8 1195.42  5816.9 1207.55  5887.9 1238.60  5935.6 1262.80  5957.7 1276.19
#Mann=5,-1,0
  4387.0    0.08       0  4899.5    0.14       0  4969.1    0.04       0
  5025.2    0.08       0  5784.8    0.14       0
#XS Ineff=2,0
       0                 5029.10    0.00 1189.60
Permanent Ineff=
       F       F
Bank Sta=4969.1,5025.2
XS Rating Curve= 0
Exp/Cntr=0.3,0.1

Type RM Length L Ch R = 1,178998,503,503,503
BEGIN DESCRIPTION:
Fisher River 358.0
END DESCRIPTION:
XS GIS Cut Line= 4
      1462602.55       994079.44      1462447.14       993736.61
      1462387.72       993517.22      1462419.71       992891.04
#Sta/Elev= 30
  4539.7 1259.87  4559.1 1253.31  4654.8 1214.52  4694.0 1201.66  4722.1 1194.03
  4783.5 1186.09  4818.4 1184.42  4884.2 1185.46  4924.5 1184.40  4960.1 1185.36
  4972.7 1176.38  4976.9 1171.38  5033.5 1171.38  5035.6 1176.38  5037.8 1177.90
  5042.2 1186.72  5267.4 1181.41  5481.2 1180.79  5500.5 1179.70  5521.4 1180.65
  5528.2 1176.38  5537.5 1180.43  5620.2 1181.79  5655.9 1185.12  5657.0 1185.27
  5671.7 1204.78  5683.6 1217.77  5719.5 1248.92  5757.4 1273.29  5770.4 1279.51
#Mann=6,-1,0
  4539.7    0.14       0  4694.0    0.08       0  4924.5    0.14       0
  4972.7    0.04       0  5035.6    0.08       0  5655.9    0.14       0
#XS Ineff=2,0
       0                 5042.20    0.00 1186.72
Permanent Ineff=
       F       F
Bank Sta=4972.7,5035.6
XS Rating Curve= 0
Exp/Cntr=0.3,0.1

Type RM Length L Ch R = 1,178495,485,485,485
BEGIN DESCRIPTION:
Fisher River 357.0
END DESCRIPTION:
XS GIS Cut Line= 4
      1463013.86       993521.78      1462803.64       993434.95
      1462748.79       993297.83      1462716.79       992977.85
#Sta/Elev= 30
  4694.9 1279.97  4745.6 1271.47  4801.7 1256.28  4844.0 1237.49  4864.6 1226.31
  4889.8 1215.72  4924.0 1205.65  4929.4 1202.53  4959.5 1196.74  4961.2 1193.80
  4967.6 1174.44  4968.5 1173.82  4969.7 1168.82  5021.9 1168.82  5023.8 1173.82
  5047.2 1173.99  5068.0 1176.46  5105.2 1173.82  5134.4 1176.34  5144.8 1183.26
  5157.0 1187.90  5168.4 1194.07  5183.9 1208.36  5188.0 1209.62  5194.3 1215.05
  5202.6 1217.16  5229.9 1216.84  5255.2 1220.45  5339.4 1237.46  5391.6 1251.63
#Mann=3,-1,0
  4694.9    0.14       0  4968.5    0.04       0  5023.8    0.14       0
Bank Sta=4968.5,5023.8
XS Rating Curve= 0
Exp/Cntr=0.3,0.1

Type RM Length L Ch R = 1,178010,499,499,499
BEGIN DESCRIPTION:
Fisher River 356.0
END DESCRIPTION:
XS GIS Cut Line= 4
      1463301.81       993311.52      1463146.43       993046.45
      1462949.90       992968.75      1462785.37       992767.67
#Sta/Elev= 30
  4628.4 1296.08  4676.9 1285.77  4755.8 1264.38  4857.5 1229.36  4878.1 1215.73
  4920.5 1196.60  4926.0 1194.69  4935.7 1189.43  4947.6 1181.89  4960.6 1171.96
  4969.9 1166.96  5022.2 1166.96  5029.5 1171.96  5052.5 1187.66  5092.8 1206.01
  5117.2 1213.98  5139.7 1231.06  5147.0 1233.85  5150.0 1236.51  5167.5 1241.93
  5188.5 1252.47  5202.1 1256.00  5206.8 1256.30  5241.1 1263.38  5311.6 1269.15
  5326.7 1271.88  5333.1 1274.51  5354.6 1280.05  5391.7 1289.43  5406.8 1292.31
#Mann=3,-1,0
  4628.4    0.14       0  4960.6    0.04       0  5029.5    0.14       0
Bank Sta=4960.6,5029.5
XS Rating Curve= 0
Exp/Cntr=0.3,0.1

Type RM Length L Ch R = 1,177511,518,518,518
BEGIN DESCRIPTION:
Fisher River 355.0
END DESCRIPTION:
XS GIS Cut Line= 3
      1463585.21       993041.91      1463448.09       992717.37
      1463187.57       992260.33
#Sta/Elev= 30
  4573.4 1238.31  4650.5 1212.69  4691.9 1201.27  4743.0 1192.48  4760.1 1188.66
  4781.2 1185.70  4820.4 1183.04  4873.2 1182.05  4891.0 1180.79  4942.1 1180.12
  4964.0 1174.75  4967.0 1172.83  4967.6 1171.08  4969.2 1171.07  4972.2 1166.07
  5035.0 1166.07  5036.5 1171.07  5043.7 1193.26  5047.9 1203.48  5051.0 1218.98
  5056.3 1220.97  5086.1 1236.07  5109.7 1245.84  5124.2 1249.84  5147.5 1250.07
  5189.0 1253.82  5230.3 1259.66  5354.3 1271.84  5381.5 1272.53  5451.8 1277.01
#Mann=3,-1,0
  4573.4    0.14       0  4969.2    0.04       0  5036.5    0.14       0
Bank Sta=4969.2,5036.5
XS Rating Curve= 0
Exp/Cntr=0.3,0.1

Type RM Length L Ch R = 1,176993,428,428,428
BEGIN DESCRIPTION:
Fisher River 354.0
END DESCRIPTION:
XS GIS Cut Line= 4
      1463978.27       992987.02      1463914.28       992502.56
      1463841.15       992356.30      1463626.36       992219.20
#Sta/Elev= 30
  4413.6 1239.98  4470.4 1215.90  4489.2 1208.43  4535.1 1192.16  4545.4 1190.29
  4569.5 1186.66  4621.7 1181.05  4647.0 1178.98  4693.4 1177.99  4717.2 1178.34
  4791.1 1177.81  4810.0 1178.22  4904.4 1178.01  4947.1 1178.80  4956.2 1173.10
  4956.5 1170.51  4958.2 1170.51  4961.3 1165.51  5032.2 1165.51  5034.7 1170.51
  5053.2 1176.25  5065.1 1178.18  5071.0 1178.16  5128.0 1178.04  5150.2 1178.99
  5192.2 1182.82  5231.9 1189.52  5257.8 1193.00  5290.4 1196.37  5320.6 1198.70
#Mann=6,-1,0
  4413.6    0.08       0  4810.0    0.14       0  4958.2    0.04       0
  5034.7    0.14       0  5071.0    0.08       0  5257.8    0.14       0
Bank Sta=4958.2,5034.7
XS Rating Curve= 0
Exp/Cntr=0.3,0.1

Type RM Length L Ch R = 1,176565,566,566,566
BEGIN DESCRIPTION:
Fisher River 353.0
END DESCRIPTION:
XS GIS Cut Line= 4
      1464522.16       991917.54      1464330.20       992104.92
      1463946.28       992278.60      1463603.52       992150.64
#Sta/Elev= 30
  4580.9 1263.01  4614.2 1255.55  4653.0 1234.28  4658.2 1226.74  4689.1 1188.41
  4697.8 1182.57  4713.3 1174.22  4778.1 1174.86  4876.7 1175.63  4911.0 1175.73
  4933.8 1174.57  4958.1 1170.60  4960.3 1169.05  4975.3 1167.65  4977.8 1162.65
  5067.1 1162.65  5068.9 1167.65  5092.0 1177.57  5095.7 1177.94  5114.2 1177.13
  5173.7 1176.61  5261.7 1177.31  5284.8 1176.91  5353.8 1177.33  5401.3 1179.79
  5466.4 1189.73  5487.2 1191.75  5529.7 1194.82  5608.4 1199.01  5636.4 1201.55
#Mann=6,-1,0
  4580.9    0.14       0  4778.1    0.08       0  4876.7    0.14       0
  4975.3    0.04       0  5068.9    0.14       0  5284.8    0.08       0
#XS Ineff=2,0
       0                 5095.70    0.00 1177.94
Permanent Ineff=
       F       F
Bank Sta=4975.3,5068.9
XS Rating Curve= 0
Exp/Cntr=0.3,0.1

Type RM Length L Ch R = 1,175999,498,498,498
BEGIN DESCRIPTION:
Fisher River 352.0
END DESCRIPTION:
XS GIS Cut Line= 5
      1464343.95       991784.96      1464151.95       991894.68
      1463914.28       991873.19      1463763.45       991891.48
      1463512.10       992072.90
#Sta/Elev= 30
  4459.4 1233.19  4502.0 1226.43  4516.0 1225.74  4573.3 1219.39  4694.0 1213.62
  4717.0 1208.99  4779.7 1192.19  4793.3 1189.49  4809.4 1188.27  4832.9 1183.89
  4863.7 1181.32  4900.8 1178.27  4929.3 1174.79  4949.3 1174.88  4962.2 1173.76
  4963.6 1171.78  4970.5 1166.36  4977.8 1161.36  5022.2 1161.36  5028.5 1166.36
  5032.4 1166.40  5034.3 1169.18  5039.3 1173.32  5097.6 1174.56  5160.7 1176.39
  5190.2 1179.00  5204.0 1180.59  5261.4 1196.08  5285.7 1198.43  5381.1 1208.02
#Mann=7,-1,0
  4459.4    0.08       0  4863.7    0.14       0  4970.5    0.04       0
  5028.5    0.14       0  5097.6    0.08       0  5190.2    0.14       0
  5285.7    0.08       0
Bank Sta=4970.5,5028.5
XS Rating Curve= 0
Exp/Cntr=0.3,0.1

Type RM Length L Ch R = 1,175501,501,501,501
BEGIN DESCRIPTION:
Fisher River 351.0
END DESCRIPTION:
XS GIS Cut Line= 4
      1464321.07       991653.81      1463690.32       991416.14
      1463566.92       991475.56      1463082.43       991736.08
#Sta/Elev= 30
  4262.0 1237.92  4300.5 1231.12  4341.5 1221.39  4411.5 1201.32  4492.8 1181.52
  4558.4 1176.24  4618.7 1175.41  4730.8 1174.54  4754.1 1170.32  4827.5 1171.78
  4848.6 1169.71  4897.8 1174.05  4957.3 1174.04  4963.9 1172.68  4974.9 1166.14
  4975.3 1164.65  4977.8 1159.65  5030.5 1159.65  5030.6 1164.65  5032.4 1164.75
  5044.9 1175.22  5055.0 1173.30  5123.3 1173.28  5317.4 1172.81  5397.4 1175.84
  5462.5 1182.76  5545.1 1198.50  5570.3 1205.78  5585.7 1212.81  5623.1 1225.84
#Mann=6,-1,0
  4262.0     0.1       0  4618.7    0.14       0  4975.3    0.04       0
  5030.6    0.14       0  5123.3    0.08       0  5545.1    0.14       0
#XS Ineff=2,0
    0.00 4952.40 1174.08 5044.90    0.00 1175.22
Permanent Ineff=
       F       F
Bank Sta=4975.3,5030.6
XS Rating Curve= 0
Exp/Cntr=0.3,0.1

Type RM Length L Ch R = 1,175000,493,493,493
BEGIN DESCRIPTION:
Fisher River 350.0
END DESCRIPTION:
XS GIS Cut Line= 4
      1464380.50       991630.97      1463919.28       991402.41
      1463900.57       991032.21      1463640.03       990968.22
#Sta/Elev= 30
  4376.4 1247.11  4439.2 1236.20  4498.9 1223.47  4598.1 1196.00  4619.6 1193.47
  4625.6 1193.89  4640.5 1188.22  4667.0 1182.74  4702.2 1178.26  4744.3 1175.02
  4936.0 1172.82  4954.2 1170.95  4957.6 1169.35  4965.0 1162.85  4977.8 1157.85
  5022.2 1157.85  5027.9 1162.85  5029.6 1162.86  5034.1 1171.69  5036.9 1172.07
  5098.7 1173.33  5116.2 1167.77  5129.1 1182.66  5140.5 1184.88  5215.7 1189.12
  5279.0 1189.40  5385.8 1192.82  5441.8 1196.56  5481.2 1201.99  5530.1 1211.71
#Mann=4,-1,0
  4376.4     0.1       0  4965.0    0.04       0  5027.9    0.14       0
  5279.0    0.08       0
#XS Ineff=2,0
       0                 5067.60    0.00 1173.43
Permanent Ineff=
       F       F
Bank Sta=4965,5027.9
XS Rating Curve= 0
Exp/Cntr=0.3,0.1

Type RM Length L Ch R = 1,174507,517,517,517
BEGIN DESCRIPTION:
Fisher River 349.0
END DESCRIPTION:
XS GIS Cut Line= 4
      1464449.03       991585.22      1464325.63       991036.78
      1464170.23       990899.67      1463640.00       990885.95
#Sta/Elev= 30
  4340.0 1246.48  4375.5 1236.39  4469.8 1205.42  4502.9 1196.95  4532.9 1191.36
  4645.8 1177.80  4697.5 1173.30  4746.2 1170.58  4816.8 1170.06  4935.5 1170.53
  4964.8 1164.01  4967.4 1161.89  4971.9 1157.10  5022.2 1157.10  5024.7 1162.10
  5026.9 1162.11  5029.9 1167.60  5050.3 1174.63  5055.9 1173.91  5074.7 1175.97
  5107.5 1176.71  5122.5 1178.15  5182.6 1182.35  5261.1 1183.52  5417.7 1188.21
  5504.4 1192.56  5575.1 1197.72  5580.1 1199.53  5616.9 1205.74  5639.8 1211.06
#Mann=5,-1,0
  4340.0    0.08       0  4816.8    0.14       0  4967.4    0.04       0
  5024.7    0.14       0  5122.5    0.08       0
Bank Sta=4967.4,5024.7
XS Rating Curve= 0
Exp/Cntr=0.3,0.1

Type RM Length L Ch R = 1,173990,456,456,456
BEGIN DESCRIPTION:
Fisher River 348.0
END DESCRIPTION:
XS GIS Cut Line= 4
      1464750.69       991548.68      1464732.41       990917.95
      1464714.13       990675.71      1464001.15       990186.68
#Sta/Elev= 30
  4285.7 1237.98  4350.9 1216.31  4408.5 1200.61  4424.0 1195.40  4444.2 1193.34
  4462.7 1188.16  4474.9 1187.94  4505.8 1182.41  4570.5 1176.43  4688.8 1171.49
  4858.2 1168.83  4921.4 1169.51  4952.6 1171.00  4975.3 1161.33  4977.8 1156.33
  5022.2 1156.33  5024.7 1161.33  5036.0 1169.36  5107.7 1167.73  5191.8 1168.01
  5204.8 1166.55  5233.0 1166.23  5266.0 1167.64  5398.6 1168.22  5578.5 1172.51
  5700.7 1177.68  5744.8 1178.62  5770.7 1177.79  5813.3 1180.06  6024.2 1185.59
#Mann=4,-1,0
  4285.7    0.08       0  4858.2    0.14       0  4975.3    0.04       0
  5024.7    0.08       0
Bank Sta=4975.3,5024.7
XS Rating Curve= 0
Exp/Cntr=0.3,0.1

Type RM Length L Ch R = 1,173534,482,482,482
BEGIN DESCRIPTION:
Fisher River 347.0
END DESCRIPTION:
XS GIS Cut Line= 3
      1465248.87       991411.54      1465093.48       990588.87
      1464056.00       990090.70
#Sta/Elev= 30
  4104.8 1226.86  4149.9 1218.20  4220.3 1200.01  4256.3 1199.05  4288.9 1187.35
  4306.4 1183.34  4355.6 1177.06  4397.1 1174.04  4485.3 1171.23  4784.0 1169.12
  4879.8 1167.68  4957.5 1168.59  4969.9 1167.40  4973.1 1160.73  4975.3 1160.73
  4977.8 1155.73  5022.2 1155.73  5024.7 1160.73  5029.0 1160.73  5031.3 1169.02
  5060.2 1166.82  5210.6 1167.14  5248.5 1165.50  5282.0 1167.14  5438.0 1167.62
  5624.1 1171.67  5728.5 1176.84  5802.6 1178.40  5823.7 1176.99  6092.9 1185.40
#Mann=5,-1,0
  4104.8    0.08       0  4784.0    0.14       0  4975.3    0.04       0
  5024.7    0.14       0  5210.6    0.08       0
Bank Sta=4975.3,5024.7
XS Rating Curve= 0
Exp/Cntr=0.3,0.1

Type RM Length L Ch R = 1,173052,444,444,444
BEGIN DESCRIPTION:
Fisher River 346.0
END DESCRIPTION:
XS GIS Cut Line= 4
      1465984.75       990844.84      1465376.86       990214.08
      1465248.88       990122.67      1464101.67       989999.27
#Sta/Elev= 30
  4031.3 1236.87  4072.2 1228.96  4097.0 1218.01  4136.0 1180.72  4161.2 1180.89
  4186.2 1176.60  4227.9 1172.95  4411.9 1168.40  4524.7 1166.78  4804.6 1166.06
  4859.5 1167.51  4899.6 1164.72  4969.7 1166.73  4971.5 1164.24  4973.8 1159.07
  4975.3 1158.06  4977.8 1153.06  5022.2 1153.06  5024.7 1158.06  5028.6 1159.06
  5029.3 1163.47  5030.8 1167.73  5064.6 1166.56  5188.0 1166.29  5199.3 1165.12
  5724.6 1169.49  5884.2 1174.29  5907.4 1177.00  5940.7 1178.76  6218.4 1184.80
#Mann=5,-1,0
  4031.3    0.08       0  4804.6    0.14       0  4975.3    0.04       0
  5024.7    0.14       0  5199.3    0.08       0
Bank Sta=4975.3,5024.7
XS Rating Curve= 0
Exp/Cntr=0.5,0.3

Type RM Length L Ch R = 1,172608,194,194,194
BEGIN DESCRIPTION:
Haystack Rd - US
END DESCRIPTION:
XS GIS Cut Line= 6
      1466399.88       990311.43      1465975.78       990179.81
      1465829.52       990080.35      1465422.93       989700.08
      1465007.56       989670.83      1464208.94       989741.04
#Sta/Elev= 30
  4016.5 1232.42  4065.2 1196.72  4100.5 1177.06  4125.0 1172.32  4150.1 1171.42
  4201.4 1174.73  4213.6 1173.35  4225.0 1169.30  4240.3 1168.82  4240.9 1167.45
  4250.3 1170.78  4285.1 1168.24  4490.3 1165.43  4795.1 1164.90  4867.1 1166.27
  4954.7 1164.36  4967.5 1161.91  4975.0 1151.71  5033.7 1151.71  5034.7 1161.78
  5038.8 1168.22  5058.6 1164.95  5150.0 1164.62  5181.8 1162.99  5244.7 1165.64
  5301.8 1165.29  5591.2 1166.03  5960.4 1171.44  5986.7 1170.48  6415.6 1180.28
#Mann=4,-1,0
  4016.5    0.08       0  4967.5    0.04       0  5034.7    0.14       0
  5301.8    0.08       0
#XS Ineff=2,0
    0.00 4900.00 1173.40 5100.00    0.00 1173.40
Permanent Ineff=
       F       F
Bank Sta=4967.5,5034.7
XS Rating Curve= 0
Exp/Cntr=0.5,0.3

Type RM Length L Ch R =3,172489,,,
BEGIN DESCRIPTION:
Haystack Rd - TOR
Structure ID: LDS_FR_12
Approximate Survey Structure
END DESCRIPTION:
Bridge Culvert--1,0,-1,-1,0
Deck Dist Width WeirC Skew NumUp NumDn MinLoCord MaxHiCord MaxSubmerge Is_Ogee
104,30,3,,24,24,,,0.95,0,1,1,,,
  4193.3  4284.1  4910.0  4910.0  5090.0  5090.0  5101.2  5203.3  5240.3  5387.5
  5466.5  5536.5  5608.6  5638.1  5681.4  5739.0  5784.9  5825.9  5899.1  5951.5
  6027.2  6055.9  6419.3  6426.0
 1174.35 1173.40 1173.40 1173.40 1173.40 1173.40 1173.40 1174.48 1175.09 1179.66
 1181.89 1184.61 1185.94 1186.44 1186.57 1186.19 1185.68 1184.44 1182.72 1182.27
 1182.06 1182.25 1189.36 1189.60
 1131.71 1131.71 1131.71 1168.90 1168.90 1131.71 1131.71 1131.71 1131.71 1131.71
 1131.71 1131.71 1131.71 1131.71 1131.71 1131.71 1131.71 1131.71 1131.71 1131.71
 1131.71 1131.71 1131.71 1131.71
  4193.3  4284.1  4910.0  4910.0  5090.0  5090.0  5101.2  5203.3  5240.3  5387.5
  5466.5  5536.5  5608.6  5638.1  5681.4  5739.0  5784.9  5825.9  5899.1  5951.5
  6027.2  6055.9  6419.3  6426.0
 1174.35 1173.40 1173.40 1173.40 1173.40 1173.40 1173.40 1174.48 1175.09 1179.66
 1181.89 1184.61 1185.94 1186.44 1186.57 1186.19 1185.68 1184.44 1182.72 1182.27
 1182.06 1182.25 1189.36 1189.60
 1131.71 1131.71 1131.71 1168.90 1168.90 1131.71 1131.71 1131.71 1131.71 1131.71
 1131.71 1131.71 1131.71 1131.71 1131.71 1131.71 1131.71 1131.71 1131.71 1131.71
 1131.71 1131.71 1131.71 1131.71
Pier Skew, UpSta & Num, DnSta & Num=,4955,2,4955,2,0,0,0,0,0
       3       3
 1164.30 1168.90
       3       3
 1163.73 1168.90
Pier Skew, UpSta & Num, DnSta & Num=,5045,2,5045,2,0,0,0,0,0
       3       3
 1166.76 1168.90
       3       3
 1163.30 1168.90
BR Coef=1,1,0,1.25,0,,,0.8,0,2,0,
WSPro=,,,, 1 ,,,, 0 ,,,, 0 ,,,,-1 ,-1 ,-1 , 0 , 0 , 0 , 0 , 0
BC Design=,,0,,0,,,,,,

Type RM Length L Ch R = 1,172414,463,463,463
BEGIN DESCRIPTION:
Haystack Rd - DS
END DESCRIPTION:
XS GIS Cut Line= 6
      1466448.32       990245.38      1465942.83       989924.51
      1465683.51       989643.21      1465516.81       989498.99
      1465116.51       989274.00      1464945.10       988720.21
#Sta/Elev= 30
  4070.0 1215.47  4099.7 1208.88  4129.2 1197.63  4155.8 1183.37  4175.4 1179.04
  4218.3 1175.57  4237.8 1171.41  4248.8 1172.66  4333.8 1168.63  4668.7 1164.75
  4816.2 1164.46  4888.6 1166.10  4967.5 1162.66  4975.0 1151.46  5028.4 1151.46
  5037.2 1162.66  5164.5 1164.71  5289.4 1174.81  5332.7 1175.80  5352.2 1179.84
  5381.1 1183.34  5501.6 1187.36  5596.4 1188.50  5917.6 1187.53  6055.1 1189.67
  6157.4 1193.61  6172.4 1192.98  6201.1 1195.88  6229.7 1214.60  6311.1 1240.28
#Mann=5,-1,0
  4070.0    0.08       0  4967.5    0.04       0  5037.2    0.14       0
  5352.2    0.08       0  6157.4    0.14       0
#XS Ineff=2,0
    0.00 4900.00 1171.50 5100.00    0.00 1171.50
Permanent Ineff=
       F       F
Bank Sta=4967.5,5037.2
XS Rating Curve= 0
Exp/Cntr=0.5,0.3

Type RM Length L Ch R = 1,171951,445,445,445
BEGIN DESCRIPTION:
Fisher River 344.0
END DESCRIPTION:
XS GIS Cut Line= 3
      1466892.23       989911.33      1465784.60       989208.07
      1464962.65       988693.80
#Sta/Elev= 30
  3810.6 1227.61  3831.9 1215.04  3863.8 1214.99  3890.9 1201.92  3961.0 1179.92
  4006.0 1176.86  4028.4 1171.60  4089.8 1167.81  4157.2 1169.17  4620.1 1162.26
  4691.7 1163.94  4898.8 1160.81  4925.8 1162.46  4960.9 1159.67  4967.2 1155.53
  4977.8 1150.53  5022.2 1150.53  5024.7 1155.53  5029.3 1155.57  5042.0 1163.76
  5250.8 1161.19  5302.3 1164.83  5333.2 1172.94  5625.6 1177.14  5854.5 1188.43
  5919.1 1198.43  5951.3 1196.97  5985.2 1214.70  6030.9 1231.42  6092.2 1245.50
#Mann=3,-1,0
  3810.6    0.08       0  4967.2    0.04       0  5024.7    0.08       0
Bank Sta=4967.2,5024.7
XS Rating Curve= 0
Exp/Cntr=0.3,0.1

Type RM Length L Ch R = 1,171506,509,509,509
BEGIN DESCRIPTION:
Fisher River 343.0
END DESCRIPTION:
XS GIS Cut Line= 4
      1466905.42       989177.30      1466158.21       988904.79
      1465969.21       988887.21      1465243.98       988500.42
#Sta/Elev= 30
  4112.9 1217.54  4147.8 1211.81  4163.9 1206.90  4195.5 1199.52  4288.8 1169.92
  4324.9 1167.64  4587.1 1160.54  4917.6 1160.85  4929.0 1157.63  4937.3 1156.88
  4954.0 1160.48  4965.0 1154.81  4977.8 1149.81  5022.2 1149.81  5024.7 1154.81
  5024.8 1162.74  5053.7 1161.51  5165.6 1160.50  5278.4 1161.29  5290.8 1163.19
  5310.7 1172.02  5423.3 1174.17  5595.4 1175.51  5720.5 1181.92  5803.4 1184.31
  5867.8 1191.72  5879.0 1194.15  5895.4 1202.11  5901.1 1203.19  5920.0 1203.39
#Mann=3,-1,0
  4112.9    0.08       0  4965.0    0.04       0  5024.7    0.08       0
Bank Sta=4965,5024.7
XS Rating Curve= 0
Exp/Cntr=0.3,0.1

Type RM Length L Ch R = 1,170997,491,491,491
BEGIN DESCRIPTION:
Fisher River 342.0
END DESCRIPTION:
XS GIS Cut Line= 4
      1466931.80       989159.74      1466404.35       988531.19
      1466180.18       988386.14      1465494.52       987792.77
#Sta/Elev= 30
  4085.8 1223.80  4111.4 1220.16  4159.4 1204.94  4194.6 1187.60  4219.3 1170.11
  4260.1 1168.15  4290.6 1163.08  4594.5 1158.74  4768.8 1160.49  4815.9 1158.94
  4968.7 1161.61  4975.3 1153.53  4977.8 1148.53  5038.7 1148.53  5038.8 1153.53
  5043.3 1153.58  5043.4 1157.04  5050.2 1166.61  5097.0 1171.43  5218.8 1171.79
  5616.4 1169.60  5632.8 1171.50  5748.5 1172.61  5877.6 1178.13  5945.6 1183.76
  5991.8 1194.84  6036.2 1198.77  6046.1 1201.08  6066.7 1210.03  6080.1 1211.15
#Mann=4,-1,0
  4085.8    0.08       0  4975.3    0.04       0  5038.8    0.15       0
  5218.8    0.08       0
Bank Sta=4975.3,5038.8
XS Rating Curve= 0
Exp/Cntr=0.3,0.1

Type RM Length L Ch R = 1,170506,487,487,487
BEGIN DESCRIPTION:
Fisher River 341.0
END DESCRIPTION:
XS GIS Cut Line= 4
      1467380.14       987735.62      1466606.53       988069.68
      1466443.90       988008.14      1466413.14       987507.12
#Sta/Elev= 30
  4043.1 1189.44  4112.7 1183.84  4261.2 1177.39  4455.5 1178.71  4492.6 1173.58
  4505.3 1173.65  4520.8 1169.75  4545.5 1155.72  4555.1 1155.34  4560.5 1157.31
  4564.3 1153.51  4568.3 1157.11  4869.6 1158.99  4919.4 1159.19  4939.0 1155.96
  4960.1 1155.86  4975.3 1151.60  4977.8 1146.60  5022.2 1146.60  5024.7 1151.60
  5032.3 1159.33  5089.4 1158.78  5293.2 1160.13  5322.3 1160.11  5351.2 1167.27
  5401.1 1187.09  5428.7 1202.42  5444.4 1209.16  5469.4 1217.00  5561.6 1234.72
#Mann=6,-1,0
  4043.1    0.08       0  4869.6    0.14       0  4975.3    0.04       0
  5024.7    0.08       0  5089.4    0.08       0  5293.2    0.14       0
Bank Sta=4975.3,5024.7
XS Rating Curve= 0
Exp/Cntr=0.3,0.1

Type RM Length L Ch R = 1,170019,529,529,529
BEGIN DESCRIPTION:
Fisher River 340.0
END DESCRIPTION:
XS GIS Cut Line= 4
      1467384.48       987709.25      1466892.23       987647.72
      1466492.25       987616.96      1466439.52       987507.09
#Sta/Elev= 30
  4325.1 1190.12  4383.0 1184.88  4462.7 1180.67  4577.0 1177.70  4711.0 1176.78
  4850.3 1171.98  4870.6 1171.04  4883.0 1167.97  4891.1 1165.13  4901.5 1159.64
  4906.8 1157.78  4930.1 1155.68  4978.8 1156.46  4987.7 1155.76  4996.4 1152.67
  4999.5 1150.46  5001.2 1145.46  5065.4 1145.46  5067.2 1150.46  5075.7 1157.28
  5085.8 1157.90  5109.9 1156.58  5124.7 1157.02  5134.4 1155.97  5161.4 1168.01
  5197.0 1193.49  5247.2 1218.21  5284.6 1228.96  5323.7 1234.63  5344.2 1236.63
#Mann=4,-1,0
  4325.1    0.08       0  4850.3    0.14       0  4999.5    0.04       0
  5067.2    0.14       0
Bank Sta=4999.5,5067.2
XS Rating Curve= 0
Exp/Cntr=0.3,0.1

Type RM Length L Ch R = 1,169490,488,488,488
BEGIN DESCRIPTION:
Fisher River 339.0
END DESCRIPTION:
XS GIS Cut Line= 5
      1467375.74       987608.17      1467301.00       987581.79
      1467032.88       987309.28      1466646.09       987133.47
      1466624.11       986878.54
#Sta/Elev= 30
  4381.4 1189.31  4474.3 1183.36  4578.6 1180.08  4715.9 1171.90  4756.4 1171.34
  4808.6 1168.15  4852.9 1167.08  4860.6 1164.29  4873.4 1164.34  4916.0 1158.59
  4960.6 1156.14  4970.1 1148.30  4972.0 1148.30  4975.9 1143.30  5022.2 1143.30
  5024.7 1148.30  5024.9 1148.48  5025.6 1154.74  5028.1 1157.26  5246.4 1156.67
  5362.4 1154.55  5370.9 1170.65  5385.1 1183.01  5395.6 1194.68  5423.2 1204.25
  5435.2 1217.19  5460.0 1240.57  5497.0 1254.25  5516.8 1259.17  5523.7 1259.62
#Mann=4,-1,0
  4381.4    0.08       0  4808.6    0.14       0  4972.0    0.04       0
  5024.7    0.14       0
Bank Sta=4972,5024.7
XS Rating Curve= 0
Exp/Cntr=0.3,0.1

Type RM Length L Ch R = 1,169002,507,507,507
BEGIN DESCRIPTION:
Fisher River 338.0
END DESCRIPTION:
XS GIS Cut Line= 3
      1467437.25       987102.70      1467090.02       986777.44
      1466843.89       986729.10
#Sta/Elev= 30
  4651.4 1210.37  4686.5 1200.48  4707.4 1196.29  4776.7 1179.63  4817.8 1173.72
  4872.0 1169.45  4886.2 1166.52  4902.4 1165.06  4942.0 1156.27  4956.6 1154.65
  4964.4 1154.88  4973.3 1149.38  4975.3 1147.12  4977.8 1142.12  5034.4 1142.12
  5034.5 1147.12  5035.1 1150.27  5045.5 1155.10  5074.3 1155.40  5132.0 1153.22
  5139.7 1154.23  5160.8 1163.15  5174.7 1166.55  5181.9 1166.58  5216.8 1176.07
  5226.0 1176.99  5268.4 1193.70  5298.8 1203.04  5326.3 1209.36  5378.0 1217.10
#Mann=3,-1,0
  4651.4    0.14       0  4975.3    0.04       0  5034.5    0.14       0
Bank Sta=4975.3,5034.5
XS Rating Curve= 0
Exp/Cntr=0.3,0.1

Type RM Length L Ch R = 1,168495,495,495,495
BEGIN DESCRIPTION:
Fisher River 337.0
END DESCRIPTION:
XS GIS Cut Line= 4
      1467709.72       986641.17      1467279.02       986412.63
      1467081.23       986447.79      1466835.10       986584.04
#Sta/Elev= 30
  4422.3 1190.11  4459.1 1184.84  4596.7 1172.75  4625.3 1170.92  4683.3 1169.07
  4747.2 1167.95  4785.4 1164.63  4831.5 1157.61  4874.2 1153.71  4911.8 1153.31
  4945.4 1155.21  4953.8 1154.35  4963.8 1154.46  4975.3 1145.96  4977.8 1140.96
  5022.2 1140.96  5024.7 1145.96  5026.5 1145.99  5029.4 1151.43  5039.6 1154.14
  5051.3 1151.95  5067.7 1151.00  5082.8 1153.09  5110.8 1154.19  5161.1 1160.73
  5192.7 1170.44  5255.4 1180.04  5303.4 1188.33  5321.7 1193.32  5392.1 1208.64
#Mann=3,-1,0
  4422.3    0.14       0  4975.3    0.04       0  5024.7    0.09       0
Bank Sta=4975.3,5024.7
XS Rating Curve= 0
Exp/Cntr=0.3,0.1

Type RM Length L Ch R = 1,168000,486,486,486
BEGIN DESCRIPTION:
Fisher River 336.0
END DESCRIPTION:
XS GIS Cut Line= 3
      1467740.54       986597.25      1467286.50       985969.55
      1466843.92       985362.20
#Sta/Elev= 30
  4225.3 1189.45  4266.4 1184.01  4373.2 1173.52  4474.3 1169.58  4534.2 1167.73
  4581.7 1164.72  4628.0 1157.92  4666.8 1155.94  4838.7 1153.01  4888.0 1151.65
  4949.7 1154.35  4960.0 1153.75  4973.8 1145.17  4976.3 1140.17  5031.3 1140.17
  5033.9 1145.17  5035.5 1145.18  5036.2 1149.31  5037.6 1152.66  5085.0 1153.30
  5107.0 1157.30  5152.1 1168.36  5174.2 1170.63  5470.2 1177.16  5523.9 1179.15
  5540.2 1185.42  5567.8 1184.36  5574.2 1185.53  5670.7 1218.15  5751.5 1237.95
#Mann=6,-1,0
  4225.3    0.08       0  4474.3    0.14       0  4534.2    0.08       0
  4838.7    0.14       0  4973.8    0.04       0  5033.9    0.08       0
Bank Sta=4973.8,5033.9
XS Rating Curve= 0
Exp/Cntr=0.3,0.1

Type RM Length L Ch R = 1,167514,512,512,512
BEGIN DESCRIPTION:
Fisher River 335.0
END DESCRIPTION:
XS GIS Cut Line= 3
      1468303.11       985964.30      1467274.62       985537.96
      1466962.57       985322.60
#Sta/Elev= 30
  4308.1 1175.48  4438.8 1168.18  4519.4 1166.13  4627.4 1160.80  4683.6 1157.61
  4726.1 1150.95  4829.3 1149.87  4859.6 1148.39  4892.9 1149.00  4924.0 1152.23
  4955.0 1145.96  4973.8 1145.07  4976.3 1140.07  5023.7 1140.07  5026.2 1145.07
  5027.5 1145.07  5028.8 1150.43  5038.4 1151.43  5069.5 1152.50  5156.0 1151.49
  5270.3 1151.87  5313.2 1153.75  5356.3 1158.51  5368.9 1160.53  5381.2 1164.41
  5617.0 1176.80  5639.6 1185.20  5687.8 1186.18  5741.4 1207.48  5800.6 1226.13
#Mann=5,-1,0
  4308.1    0.08       0  4627.4    0.14       0  4973.8    0.04       0
  5026.2    0.14       0  5156.0    0.08       0
Bank Sta=4973.8,5026.2
XS Rating Curve= 0
Exp/Cntr=0.3,0.1

Type RM Length L Ch R = 1,167002,518,518,518
BEGIN DESCRIPTION:
Fisher River 334.0
END DESCRIPTION:
XS GIS Cut Line= 4
      1468333.92       985946.77      1468048.20       985362.14
      1467665.81       985094.03      1467015.31       984948.98
#Sta/Elev= 30
  4240.3 1175.95  4278.0 1173.25  4356.1 1170.55  4409.9 1167.39  4577.1 1162.95
  4597.4 1161.33  4667.0 1150.41  4700.9 1148.92  4854.4 1149.96  4939.7 1149.73
  4957.4 1150.95  4973.8 1144.35  4976.3 1139.35  5044.9 1139.35  5047.9 1144.35
  5049.7 1144.35  5076.0 1156.09  5088.3 1159.02  5113.0 1166.94  5173.9 1169.73
  5266.4 1172.71  5584.5 1172.95  5613.6 1172.09  5637.8 1173.45  5731.5 1174.43
  5815.0 1176.90  5940.9 1182.22  5976.5 1188.42  6006.6 1187.24  6024.5 1189.47
#Mann=5,-1,0
  4240.3    0.08       0  4854.4    0.14       0  4973.8    0.04       0
  5047.9    0.14       0  5173.9    0.08       0
Bank Sta=4973.8,5047.9
XS Rating Curve= 0
Exp/Cntr=0.3,0.1

Type RM Length L Ch R = 1,166484,472,472,472
BEGIN DESCRIPTION:
Fisher River 333.0
END DESCRIPTION:
XS GIS Cut Line= 4
      1468848.13       985665.39      1468470.16       985058.87
      1467951.51       984843.49      1467015.34       984896.24
#Sta/Elev= 30
  4166.1 1195.41  4227.5 1183.98  4281.6 1177.36  4329.0 1171.37  4521.8 1161.98
  4570.0 1161.49  4715.1 1158.99  4767.0 1146.98  4928.8 1147.39  4952.2 1148.61
  4958.5 1150.17  4968.9 1147.96  4973.8 1143.64  4976.3 1138.64  5054.4 1138.64
  5058.2 1143.64  5086.0 1150.81  5214.7 1149.35  5232.1 1152.67  5253.4 1159.74
  5344.7 1165.31  5392.8 1164.76  5413.6 1167.33  5491.9 1169.15  6125.1 1174.90
  6307.9 1183.52  6320.3 1184.37  6338.4 1188.06  6366.4 1188.55  6380.0 1191.01
#Mann=7,-1,0
  4166.1    0.14       0  4281.6    0.08       0  4570.0    0.14       0
  4715.1    0.08       0  4973.8    0.04       0  5058.2    0.14       0
  5344.7    0.08       0
Bank Sta=4973.8,5058.2
XS Rating Curve= 0
Exp/Cntr=0.3,0.1

Type RM Length L Ch R = 1,166012,508,508,508
BEGIN DESCRIPTION:
Fisher River 332.0
END DESCRIPTION:
XS GIS Cut Line= 4
      1469393.21       984672.07      1468667.95       984720.42
      1468215.23       984443.52      1467024.07       983977.60
#Sta/Elev= 30
  3992.4 1206.73  4015.2 1200.81  4101.1 1172.67  4148.9 1158.65  4173.3 1154.57
  4210.8 1151.44  4283.7 1147.55  4345.9 1148.00  4409.0 1146.58  4713.6 1146.58
  4871.8 1148.83  4925.1 1146.54  4934.3 1143.23  4934.5 1144.82  4945.1 1145.10
  4955.7 1142.34  4969.2 1137.34  5030.8 1137.34  5034.1 1142.34  5037.7 1159.13
  5039.6 1159.68  5056.8 1161.60  5148.4 1165.64  5199.3 1167.86  5386.3 1169.93
  5615.7 1169.04  5822.1 1171.68  6449.0 1188.05  6497.2 1191.28  6529.0 1194.96
#Mann=4,-1,0
  3992.4    0.14       0  4955.7    0.04       0  5034.1    0.14       0
  5148.4    0.08       0
Bank Sta=4955.7,5034.1
XS Rating Curve= 0
Exp/Cntr=0.3,0.1

Type RM Length L Ch R = 1,165504,511,511,511
BEGIN DESCRIPTION:
Fisher River 331.0
END DESCRIPTION:
XS GIS Cut Line= 4
      1469401.96       984628.12      1469032.76       984522.63
      1468773.44       984223.75      1467068.08       983960.04
#Sta/Elev= 30
  4327.6 1211.20  4354.9 1204.88  4408.8 1189.04  4492.4 1166.54  4550.8 1152.15
  4594.6 1147.52  4695.5 1145.37  4739.6 1143.40  4780.2 1144.66  4859.3 1143.96
  4916.7 1144.28  4944.9 1145.75  4957.4 1139.26  4970.2 1134.26  5034.2 1134.26
  5038.5 1139.26  5043.3 1156.12  5063.0 1158.37  5138.6 1159.69  5251.8 1158.59
  5307.4 1160.73  5463.9 1161.94  5661.6 1166.06  5799.9 1166.36  5847.4 1168.90
  5872.1 1168.27  5943.2 1168.91  6279.1 1174.31  6774.8 1188.47  6832.9 1192.12
#Mann=6,-1,0
  4327.6    0.14       0  4492.4    0.08       0  4859.3    0.14       0
  4957.4    0.04       0  5038.5    0.14       0  5251.8    0.08       0
Bank Sta=4957.4,5038.5
XS Rating Curve= 0
Exp/Cntr=0.3,0.1

Type RM Length L Ch R = 1,164993,497,497,497
BEGIN DESCRIPTION:
Fisher River 330.0
END DESCRIPTION:
XS GIS Cut Line= 4
      1469700.88       984166.62      1469278.90       984021.56
      1469151.44       983894.10      1467824.07       982606.29
#Sta/Elev= 30
  4495.7 1228.82  4602.5 1192.82  4646.8 1179.62  4663.9 1171.78  4673.2 1170.79
  4691.4 1160.36  4726.0 1143.95  4774.4 1142.02  4873.6 1143.94  4939.3 1144.49
  4953.7 1138.07  4966.4 1133.07  5033.8 1133.07  5038.0 1138.07  5048.5 1139.09
  5081.9 1154.11  5116.6 1157.41  5348.7 1156.95  5425.9 1158.66  5529.0 1162.71
  5610.9 1161.02  5629.1 1162.75  5886.8 1163.62  5892.9 1164.98  5958.5 1165.64
  6169.2 1164.29  6736.2 1170.59  6829.0 1175.45  6899.8 1190.12  6971.6 1200.54
#Mann=6,-1,0
  4495.7    0.14       0  4726.0    0.08       0  4873.6    0.14       0
  4953.7    0.04       0  5038.0    0.14       0  5425.9    0.08       0
Bank Sta=4953.7,5038
XS Rating Curve= 0
Exp/Cntr=0.3,0.1

Type RM Length L Ch R = 1,164496,483,483,483
BEGIN DESCRIPTION:
Fisher River 329.0
END DESCRIPTION:
XS GIS Cut Line= 4
      1469964.61       983678.74      1469555.81       983577.63
      1469278.90       983538.08      1467837.26       982588.70
#Sta/Elev= 30
  4485.2 1241.40  4522.8 1233.67  4565.6 1218.65  4602.7 1201.32  4662.5 1159.36
  4685.5 1145.08  4706.0 1139.88  4719.8 1140.98  4943.8 1144.78  4946.2 1138.87
  4954.3 1137.03  4958.5 1132.03  5029.1 1132.03  5029.2 1137.03  5034.6 1137.06
  5047.7 1146.63  5073.7 1143.41  5148.7 1145.88  5234.1 1155.54  5366.0 1160.38
  5454.6 1164.31  5553.8 1161.77  5894.4 1164.89  6243.1 1165.65  6312.7 1169.08
  6682.9 1171.79  6697.1 1174.69  6739.5 1175.82  6796.5 1188.21  6912.2 1201.92
#Mann=5,-1,0
  4485.2    0.14       0  4719.8    0.08       0  4954.3    0.04       0
  5029.2    0.14       0  5366.0    0.08       0
Bank Sta=4954.3,5029.2
XS Rating Curve= 0
Exp/Cntr=0.3,0.1

Type RM Length L Ch R = 1,164013,527,527,527
BEGIN DESCRIPTION:
Fisher River 328.0
END DESCRIPTION:
XS GIS Cut Line= 4
      1470034.88       983476.53      1469810.74       983226.01
      1469586.57       983120.52      1468158.10       982522.76
#Sta/Elev= 30
  4593.7 1205.13  4713.3 1157.48  4735.7 1144.04  4745.0 1140.66  4783.8 1140.16
  4942.9 1140.39  4955.5 1142.95  4959.7 1140.11  4961.3 1136.22  4965.0 1131.22
  5023.7 1131.22  5026.2 1136.22  5045.6 1142.58  5069.9 1141.39  5132.1 1153.60
  5278.4 1154.83  5326.1 1157.34  5414.3 1162.77  5453.4 1159.79  5546.6 1159.53
  5656.9 1159.61  5778.0 1163.18  5936.7 1162.40  6184.9 1175.21  6458.7 1174.12
  6559.0 1179.38  6593.3 1184.06  6622.9 1182.33  6657.6 1190.02  6726.1 1197.71
#Mann=5,-1,0
  4593.7    0.14       0  4783.8    0.08       0  4961.3    0.04       0
  5026.2    0.14       0  5326.1    0.08       0
Bank Sta=4961.3,5026.2
XS Rating Curve= 0
Exp/Cntr=0.3,0.1

Type RM Length L Ch R = 1,163486,494,494,494
BEGIN DESCRIPTION:
Fisher River 327.0
END DESCRIPTION:
XS GIS Cut Line= 4
      1470122.79       982830.41      1469964.57       982699.88
      1468593.23       982676.59      1468232.79       982483.19
#Sta/Elev= 30
  4715.8 1191.32  4755.1 1181.11  4792.7 1168.46  4802.9 1164.23  4830.5 1147.44
  4841.9 1146.47  4869.1 1141.81  4890.4 1140.80  4931.2 1140.78  4957.4 1143.17
  4967.9 1135.46  4976.3 1130.46  5023.7 1130.46  5026.2 1135.46  5043.7 1143.71
  5143.7 1139.87  5224.0 1141.37  5251.3 1145.93  5278.3 1144.32  5323.7 1149.47
  5495.5 1158.71  5902.3 1162.96  6194.6 1175.51  6486.9 1174.50  6558.6 1178.23
  6595.7 1184.20  6624.2 1183.47  6636.3 1184.93  6657.5 1191.17  6701.5 1196.63
#Mann=4,-1,0
  4715.8    0.14       0  4841.9    0.08       0  4967.9    0.04       0
  5026.2    0.08       0
Bank Sta=4967.9,5026.2
XS Rating Curve= 0
Exp/Cntr=0.3,0.1
