HEC-RAS study Fisher River.prj: Fisher River Limited Detail Study

--- Fisher River.g01 (geometry) --- (continued)

Type RM Length L Ch R =3,43101,,,
BEGIN DESCRIPTION:
NC Highway 268 - TOR
Structure ID: LDS_FR_04
Approximate Survey Structure
END DESCRIPTION:
Bridge Culvert--1,0,-1,-1,0
Deck Dist Width WeirC Skew NumUp NumDn MinLoCord MaxHiCord MaxSubmerge Is_Ogee
53,32,3,,41,41,,,0.95,0,1,1,,,
  4558.2  4718.5  4762.1  4805.5  4829.9  4895.0  4895.0  5105.0  5105.0  5120.4
  5130.4  5142.4  5149.3  5151.3  5161.2  5165.1  5166.4  5173.6  5183.0  5187.6
  5190.9  5196.3  5209.6  5218.3  5227.3  5231.5  5233.9  5239.8  5246.5  5253.7
  5258.2  5262.2  5275.7  5284.6  5297.8  5300.4  5317.8  5320.1  5329.0  5339.0
  5342.0
  944.20  937.61  936.12  934.98  934.74  934.60  934.60  934.60  934.60  934.64
  934.88  935.22  935.34  935.55  935.79  935.95  935.97  936.22  936.67  936.95
  937.10  937.74  938.19  938.85  939.22  939.50  939.57  939.98  940.13  940.51
  940.82  941.29  942.13  942.47  943.34  943.34  944.86  945.10  945.30  945.93
  946.25
  884.60  884.60  884.60  884.60  884.60  884.60  929.60  929.60  884.60  884.60
  884.60  884.60  884.60  884.60  884.60  884.60  884.60  884.60  884.60  884.60
  884.60  884.60  884.60  884.60  884.60  884.60  884.60  884.60  884.60  884.60
  884.60  884.60  884.60  884.60  884.60  884.60  884.60  884.60  884.60  884.60
  884.60
  4558.2  4718.5  4762.1  4805.5  4829.9  4895.0  4895.0  5105.0  5105.0  5120.4
  5130.4  5142.4  5149.3  5151.3  5161.2  5165.1  5166.4  5173.6  5183.0  5187.6
  5190.9  5196.3  5209.6  5218.3  5227.3  5231.5  5233.9  5239.8  5246.5  5253.7
  5258.2  5262.2  5275.7  5284.6  5297.8  5300.4  5317.8  5320.1  5329.0  5339.0
  5342.0
  944.20  937.61  936.12  934.98  934.74  934.60  934.60  934.60  934.60  934.64
  934.88  935.22  935.34  935.55  935.79  935.95  935.97  936.22  936.67  936.95
  937.10  937.74  938.19  938.85  939.22  939.50  939.57  939.98  940.13  940.51
  940.82  941.29  942.13  942.47  943.34  943.34  944.86  945.10  945.30  945.93
  946.25
  884.60  884.60  884.60  884.60  884.60  884.60  929.60  929.60  884.60  884.60
  884.60  884.60  884.60  884.60  884.60  884.60  884.60  884.60  884.60  884.60
  884.60  884.60  884.60  884.60  884.60  884.60  884.60  884.60  884.60  884.60
  884.60  884.60  884.60  884.60  884.60  884.60  884.60  884.60  884.60  884.60
  884.60
Pier Skew, UpSta & Num, DnSta & Num=,4947.5,2,4947.5,2,0,0,0,0,0
       3       3
  915.14  929.60
       3       3
  914.89  929.60
Pier Skew, UpSta & Num, DnSta & Num=,5052.5,2,5052.5,2,0,0,0,0,0
       3       3
  915.14  929.60
       3       3
  914.89  929.60
Abutment Skew #Up #Dn=,2,2
  4895.0  4922.0
  929.60  919.15
  4895.0  4922.0
  929.60  916.58
Abutment Skew #Up #Dn=,2,2
  5078.0  5105.0
  922.05  929.60
  5078.0  5105.0
  923.36  929.60
BR Coef=1,1,0,1.25,0,,,0.8,0,2,0,
WSPro=,,,, 1 ,,,, 0 ,,,, 0 ,,,,-1 ,-1 ,-1 , 0 , 0 , 0 , 0 , 0
BC Design=,,0,,0,,,,,,

Type RM Length L Ch R = 1,43058,559,559,559
BEGIN DESCRIPTION:
NC Highway 268 - DS
END DESCRIPTION:
XS GIS Cut Line= 4
      1504192.49       946782.35      1503767.78       946729.98
      1503499.03       946622.97      1503484.11       946540.51
#Sta/Elev= 30
  4441.6  958.56  4489.1  953.96  4539.6  945.31  4556.6  941.48  4619.2  932.93
  4635.0  933.63  4717.2  932.44  4791.5  924.57  4843.3  922.46  4855.7  924.44
  4866.3  923.66  4883.1  924.96  4907.5  919.51  4921.3  919.59  4927.8  916.76
  4943.5  913.05  4951.6  904.35  5035.3  904.35  5040.8  913.05  5068.1  920.02
  5080.4  924.99  5085.0  925.15  5104.6  929.48  5116.5  933.33  5146.3  935.90
  5155.2  935.38  5158.8  936.35  5186.9  946.84  5219.6  963.86  5242.6  973.24
#Mann=3,-1,0
  4441.6    0.14       0  4943.5    0.04       0  5040.8    0.14       0
#XS Ineff=2,0
    0.00 4885.00  932.50 5115.00    0.00  932.50
Permanent Ineff=
       F       F
Bank Sta=4943.5,5040.8
XS Rating Curve= 0
Exp/Cntr=0.5,0.3

Type RM Length L Ch R = 1,42499,1000,1000,1000
BEGIN DESCRIPTION:
Fisher River 85.0
END DESCRIPTION:
XS GIS Cut Line= 3
      1504395.57       946487.82      1504124.31       946362.27
      1503928.96       946250.64
#Sta/Elev= 30
  4632.0  940.60  4645.5  940.12  4652.6  939.19  4683.4  936.03  4717.4  931.79
  4726.1  931.21  4761.4  925.59  4778.2  923.65  4815.3  922.39  4820.8  922.41
  4823.2  921.99  4841.6  921.81  4849.1  919.89  4890.4  916.63  4906.1  917.77
  4910.5  917.64  4924.6  919.77  4930.9  919.34  4945.6  915.83  4951.0  912.96
  4957.2  908.43  4959.7  903.43  5040.3  903.43  5042.8  908.43  5044.3  908.43
  5076.8  933.01  5079.2  935.00  5082.7  937.13  5142.6  963.17  5155.9  964.99
#Mann=3,-1,0
  4632.0    0.14       0  4957.2    0.04       0  5042.8    0.14       0
Bank Sta=4957.2,5042.8
XS Rating Curve= 0
Exp/Cntr=0.3,0.1

Type RM Length L Ch R = 1,41499,498,498,498
BEGIN DESCRIPTION:
Fisher River 83.0
END DESCRIPTION:
XS GIS Cut Line= 4
      1504752.12       945523.66      1504642.05       945494.21
      1504445.19       945412.05      1504311.87       945382.60
#Sta/Elev= 30
  4772.7  956.53  4781.6  954.98  4800.9  950.96  4811.0  948.32  4823.8  945.44
  4833.8  942.57  4840.4  939.84  4852.3  939.93  4869.6  935.04  4886.6  930.74
  4909.7  924.40  4920.4  920.15  4927.8  918.22  4960.6  908.99  4962.3  906.94
  4964.7  901.94  5049.2  901.94  5053.1  906.94  5053.4  906.94  5057.3  911.64
  5070.2  918.08  5079.3  917.18  5094.6  918.98  5105.5  919.10  5124.0  918.38
  5126.2  918.43  5134.9  919.18  5171.3  931.63  5230.3  949.97  5236.5  952.05
#Mann=3,-1,0
  4772.7    0.14       0  4962.3    0.04       0  5053.1    0.14       0
Bank Sta=4962.3,5053.1
XS Rating Curve= 0
Exp/Cntr=0.3,0.1

Type RM Length L Ch R = 1,41001,420,420,420
BEGIN DESCRIPTION:
Fisher River 82.0
END DESCRIPTION:
XS GIS Cut Line= 4
      1504825.00       944975.00      1504714.91       944982.67
      1504572.30       944948.57      1504373.85       944943.91
#Sta/Elev= 30
  4812.7  970.51  4815.5  967.82  4820.3  966.78  4826.9  960.03  4845.9  948.41
  4919.2  927.92  4923.8  925.24  4932.1  925.27  4935.6  924.81  4951.6  920.02
  4955.4  919.34  4960.0  915.65  4966.6  905.50  4971.3  900.50  5049.7  900.50
  5052.7  905.50  5053.8  905.50  5059.7  914.49  5061.4  915.11  5085.3  918.17
  5111.6  923.58  5131.0  928.99  5134.7  930.39  5149.8  933.45  5162.0  936.69
  5180.9  940.13  5193.1  944.61  5218.7  952.63  5239.5  958.76  5268.2  966.27
#Mann=3,-1,0
  4812.7    0.14       0  4966.6    0.04       0  5052.7    0.14       0
Bank Sta=4966.6,5052.7
XS Rating Curve= 0
Exp/Cntr=0.3,0.1

Type RM Length L Ch R = 1,40581,300,300,300
BEGIN DESCRIPTION:
Fisher River 81.0
END DESCRIPTION:
XS GIS Cut Line= 3
      1504887.00       944533.13      1504668.40       944564.14
      1504418.88       944578.09
#Sta/Elev= 29
  4834.3  960.49  4856.9  954.92  4862.2  951.93  4871.5  947.08  4886.9  942.02
  4914.1  929.46  4917.3  926.32  4934.4  917.90  4937.1  908.69  4940.2  904.21
  4942.6  899.21  5038.7  899.21  5040.3  904.21  5040.8  904.28  5040.9  906.66
  5058.2  913.34  5105.6  916.34  5115.0  916.44  5137.0  918.68  5152.4  919.46
  5174.2  926.12  5198.2  933.09  5209.7  935.95  5219.1  936.96  5230.5  938.72
  5235.5  938.67  5259.1  946.42  5282.8  951.70  5305.0  954.14
#Mann=3,-1,0
  4834.3    0.14       0  4940.2    0.04       0  5040.3    0.14       0
Bank Sta=4940.2,5040.3
XS Rating Curve= 0
Exp/Cntr=0.5,0.3

Type RM Length L Ch R = 1,40281,72,72,72
BEGIN DESCRIPTION:
Rock Ford Road - US
END DESCRIPTION:
XS GIS Cut Line= 5
      1504899.93       944254.02      1504806.32       944199.31
      1504617.82       944300.25      1504531.48       944395.10
      1504378.54       944543.20
#Sta/Elev= 30
  4769.4  973.01  4791.4  968.25  4818.1  956.39  4828.6  950.53  4845.3  935.83
  4858.2  927.95  4863.6  926.74  4870.6  923.08  4886.3  923.74  4898.7  921.55
  4911.6  921.79  4932.1  904.90  4937.7  897.80  5046.3  897.80  5049.6  904.90
  5055.1  911.34  5056.4  912.02  5072.8  913.70  5091.6  917.58  5110.7  915.36
  5120.4  916.62  5144.0  916.70  5174.4  918.88  5201.1  922.93  5227.2  928.84
  5302.7  934.37  5377.8  942.50  5405.4  951.66  5425.7  954.76  5432.8  954.64
#Mann=3,-1,0
  4769.4    0.14       0  4932.1    0.04       0  5049.6    0.14       0
#XS Ineff=2,0
    0.00 4890.00  924.50 5110.00    0.00  924.50
Permanent Ineff=
       F       F
Bank Sta=4932.1,5049.6
XS Rating Curve= 0
Exp/Cntr=0.5,0.3

Type RM Length L Ch R =3,40244,,,
BEGIN DESCRIPTION:
Rock Ford Road - TOR
Structure ID: LDS_FR_03
Approximate Survey Structure
END DESCRIPTION:
Bridge Culvert--1,0,-1,-1,0
Deck Dist Width WeirC Skew NumUp NumDn MinLoCord MaxHiCord MaxSubmerge Is_Ogee
19.5,35,3,,10,10,,,0.95,0,1,1,,,
  4843.1  4900.0  4900.0  5100.0  5100.0  5123.7  5137.0  5146.5  5157.6  5215.7
  924.50  924.50  924.50  924.50  924.50  924.50  924.56  924.65  924.76  926.01
  877.80  877.80  920.50  920.50  877.80  877.80  877.80  877.80  877.80  877.80
  4843.1  4900.0  4900.0  5100.0  5100.0  5123.7  5137.0  5146.5  5157.6  5215.7
  924.50  924.50  924.50  924.50  924.50  924.50  924.56  924.65  924.76  926.01
  877.80  877.80  920.50  920.50  877.80  877.80  877.80  877.80  877.80  877.80
Pier Skew, UpSta & Num, DnSta & Num=,4933.3,2,4933.3,2,0,0,0,0,0
     2.5     2.5
  906.87  920.50
     2.5     2.5
  914.62  920.50
Pier Skew, UpSta & Num, DnSta & Num=,5000,2,5000,2,0,0,0,0,0
     2.5     2.5
  901.80  920.50
     2.5     2.5
  901.55  920.50
Pier Skew, UpSta & Num, DnSta & Num=,5066.7,2,5066.7,2,0,0,0,0,0
     2.5     2.5
  913.39  920.50
     2.5     2.5
  911.24  920.50
Abutment Skew #Up #Dn=,2,2
  4900.0  4925.0
  920.50  912.62
  4900.0  4925.0
  920.50  916.27
Abutment Skew #Up #Dn=,2,2
  5075.0  5100.0
  914.17  920.50
  5075.0  5100.0
  912.07  920.50
BR Coef=1,1,0,1.25,0,,,0.8,0,2,0,
WSPro=,,,, 1 ,,,, 0 ,,,, 0 ,,,,-1 ,-1 ,-1 , 0 , 0 , 0 , 0 , 0
BC Design=,,0,,0,,,,,,

Type RM Length L Ch R = 1,40209,220,220,220
BEGIN DESCRIPTION:
Rock Ford Road - DS
END DESCRIPTION:
XS GIS Cut Line= 5
      1505078.70       944040.01      1504994.03       944048.20
      1504865.91       944110.54      1504618.80       944222.34
      1504420.36       944178.93
#Sta/Elev= 30
  4589.4  985.72  4640.3  972.59  4684.4  957.66  4698.7  950.01  4720.3  936.44
  4741.1  926.28  4765.2  927.43  4815.8  924.82  4894.1  923.25  4915.2  919.53
  4932.9  912.53  4949.6  907.31  4952.5  905.49  4954.4  903.36  4954.6  902.29
  4957.5  897.55  5045.7  897.55  5046.9  902.29  5055.9  909.26  5060.4  910.20
  5083.2  912.82  5088.2  914.39  5109.2  912.13  5116.6  914.75  5151.6  921.11
  5171.5  927.46  5207.9  934.59  5216.7  937.79  5241.7  942.87  5291.3  958.26
#Mann=3,-1,0
  4589.4    0.14       0  4954.6    0.04       0  5046.9    0.14       0
#XS Ineff=2,0
    0.00 4890.00  922.50 5110.00    0.00  922.50
Permanent Ineff=
       F       F
Bank Sta=4954.6,5046.9
XS Rating Curve= 0
Exp/Cntr=0.5,0.3

Type RM Length L Ch R = 1,39989,492,492,492
BEGIN DESCRIPTION:
Fisher River 80.0
END DESCRIPTION:
XS GIS Cut Line= 4
      1505161.77       944025.13      1504824.82       943976.63
      1504667.53       943962.86      1504452.14       943953.66
#Sta/Elev= 30
  4566.1 1001.18  4589.7  999.67  4605.9  995.56  4616.1  995.03  4678.2  981.65
  4695.8  978.87  4729.5  970.87  4746.4  965.31  4794.4  933.84  4814.6  926.76
  4862.6  925.60  4920.2  920.99  4931.8  919.13  4941.0  919.77  4948.2  912.02
  4959.6  902.10  4960.7  897.10  5045.8  897.10  5047.0  902.10  5047.8  911.87
  5047.9  912.29  5067.5  915.21  5078.0  912.38  5089.0  912.11  5129.4  914.92
  5149.0  919.99  5174.9  929.58  5217.6  943.64  5244.0  950.55  5280.0  959.58
#Mann=4,-1,0
  4566.1    0.14       0  4959.6    0.04       0  5047.0    0.14       0
  5244.0    0.08       0
Bank Sta=4959.6,5047
XS Rating Curve= 0
Exp/Cntr=0.3,0.1

Type RM Length L Ch R = 1,39497,504,504,504
BEGIN DESCRIPTION:
Fisher River 79.0
END DESCRIPTION:
XS GIS Cut Line= 4
      1505286.84       943629.53      1504988.17       943540.19
      1504789.09       943466.17      1504590.01       943374.28
#Sta/Elev= 30
  4569.4  976.23  4576.2  975.64  4620.8  963.68  4642.3  956.06  4663.4  953.62
  4716.8  935.58  4736.1  925.39  4743.3  927.12  4776.6  927.58  4783.1  923.44
  4798.0  917.67  4835.1  917.66  4860.2  915.59  4882.7  915.81  4920.3  911.91
  4949.9  911.94  4953.3  908.14  4954.9  902.92  4957.2  900.71  4959.7  895.71
  5040.3  895.71  5042.8  900.71  5044.9  900.73  5047.3  903.00  5050.5  908.31
  5061.4  911.75  5187.1  917.92  5261.2  926.70  5290.1  931.67  5312.8  937.81
#Mann=3,-1,0
  4569.4    0.14       0  4957.2    0.04       0  5042.8    0.08       0
Bank Sta=4957.2,5042.8
XS Rating Curve= 0
Exp/Cntr=0.3,0.1

Type RM Length L Ch R = 1,38993,477,477,477
BEGIN DESCRIPTION:
Fisher River 78.0
END DESCRIPTION:
XS GIS Cut Line= 3
      1505401.60       943195.61      1505057.08       943034.83
      1504944.77       942945.49
#Sta/Elev= 30
  4719.5  959.72  4744.9  953.31  4805.3  935.42  4824.5  924.81  4830.7  922.44
  4839.6  922.07  4863.9  922.90  4871.1  921.46  4884.4  915.73  4889.6  916.40
  4904.3  913.99  4926.5  913.05  4938.7  910.87  4945.1  910.75  4945.4  910.03
  4956.6  904.01  4959.6  900.22  4962.8  895.22  5052.0  895.22  5054.7  900.22
  5055.8  900.22  5058.3  903.58  5061.3  906.27  5066.6  912.30  5093.8  915.41
  5127.4  918.06  5148.8  920.75  5193.0  927.85  5214.8  931.91  5243.2  934.94
#Mann=4,-1,0
  4719.5    0.08       0  4839.6    0.14       0  4959.6    0.04       0
  5054.7    0.08       0
Bank Sta=4959.6,5054.7
XS Rating Curve= 0
Exp/Cntr=0.3,0.1

Type RM Length L Ch R = 1,38516,514,514,514
BEGIN DESCRIPTION:
Fisher River 77.0
END DESCRIPTION:
XS GIS Cut Line= 4
      1505651.76       942779.60      1505496.08       942720.90
      1505304.66       942621.36      1505156.66       942575.43
#Sta/Elev= 30
  4703.6  966.10  4710.6  965.51  4757.1  957.18  4769.1  947.87  4781.7  933.06
  4801.4  933.00  4830.2  931.75  4833.4  930.83  4841.7  928.12  4867.3  922.68
  4882.4  916.24  4904.7  914.60  4938.0  909.03  4953.1  908.41  4959.8  904.80
  4961.6  900.67  4963.1  899.24  4964.0  894.24  5040.3  894.24  5040.5  899.24
  5044.3  899.47  5045.5  901.18  5047.7  901.52  5065.6  911.58  5073.4  913.75
  5083.6  912.82  5108.3  913.33  5177.8  922.23  5201.7  924.99  5240.7  926.46
#Mann=5,-1,0
  4703.6    0.08       0  4833.4    0.14       0  4963.1    0.04       0
  5040.5    0.14       0  5177.8    0.08       0
Bank Sta=4963.1,5040.5
XS Rating Curve= 0
Exp/Cntr=0.3,0.1

Type RM Length L Ch R = 1,38002,494,494,494
BEGIN DESCRIPTION:
Fisher River 76.0
END DESCRIPTION:
XS GIS Cut Line= 3
      1505457.79       942058.58      1505187.25       942403.14
      1505141.31       942569.02
#Sta/Elev= 30
  4785.7 1003.14  4804.3 1000.31  4819.0  994.94  4839.8  985.10  4884.6  952.10
  4898.8  947.56  4919.0  929.31  4928.7  924.90  4938.1  921.83  4946.7  912.81
  4948.6  897.30  4949.5  892.30  5038.9  892.30  5039.2  897.30  5042.8  909.35
  5046.7  909.88  5069.7  908.88  5081.2  907.95  5091.0  908.86  5116.8  909.65
  5127.5  912.06  5148.6  913.84  5162.2  916.91  5180.2  919.53  5198.1  919.95
  5214.3  921.32  5233.0  922.96  5275.4  925.28  5326.9  926.37  5395.9  926.49
#Mann=4,-1,0
  4785.7    0.14       0  4948.6    0.04       0  5039.2    0.14       0
  5214.3    0.08       0
Bank Sta=4948.6,5039.2
XS Rating Curve= 0
Exp/Cntr=0.3,0.1

Type RM Length L Ch R = 1,37508,488,488,488
BEGIN DESCRIPTION:
Fisher River 75.0
END DESCRIPTION:
XS GIS Cut Line= 3
      1505049.40       941844.20      1504952.44       941900.33
      1504687.01       942303.58
#Sta/Elev= 30
  4770.3  962.16  4793.8  960.38  4817.0  943.98  4825.9  940.90  4838.7  939.43
  4851.7  933.19  4859.0  926.55  4876.5  916.10  4879.8  914.92  4897.5  913.56
  4923.0  918.29  4944.7  914.25  4949.7  910.56  4957.2  896.77  4959.7  891.77
  5040.3  891.77  5042.8  896.77  5053.3  906.81  5068.0  910.26  5101.6  914.98
  5118.6  915.89  5131.4  917.41  5149.4  923.91  5204.0  947.35  5221.8  953.87
  5247.8  960.63  5254.8  961.91  5314.5  968.98  5347.8  971.82  5365.1  972.41
#Mann=4,-1,0
  4770.3    0.14       0  4957.2    0.04       0  5042.8    0.14       0
  5204.0    0.08       0
Bank Sta=4957.2,5042.8
XS Rating Curve= 0
Exp/Cntr=0.3,0.1

Type RM Length L Ch R = 1,37020,552,552,552
BEGIN DESCRIPTION:
Fisher River 74.0
END DESCRIPTION:
XS GIS Cut Line= 4
      1504544.08       941435.78      1504487.92       941619.58
      1504449.64       941872.26      1504316.92       942109.62
#Sta/Elev= 30
  4671.4  958.58  4690.1  955.82  4747.1  941.68  4757.2  940.16  4793.2  927.89
  4797.3  927.70  4817.5  923.46  4833.9  915.15  4842.1  911.92  4880.2  910.80
  4891.8  909.60  4911.4  909.27  4941.6  907.30  4955.0  907.29  4964.4  894.74
  4966.9  889.74  5034.9  889.74  5037.4  894.74  5040.1  907.58  5040.7  908.42
  5065.0  911.51  5088.1  913.37  5108.1  913.62  5145.0  928.67  5161.4  931.93
  5185.8  934.55  5195.1  936.46  5212.1  937.72  5316.1  949.63  5391.1  951.53
#Mann=3,-1,0
  4671.4    0.14       0  4964.4    0.04       0  5037.4    0.14       0
Bank Sta=4964.4,5037.4
XS Rating Curve= 0
Exp/Cntr=0.3,0.1

Type RM Length L Ch R = 1,36468,460,460,460
BEGIN DESCRIPTION:
Fisher River 73.0
END DESCRIPTION:
XS GIS Cut Line= 5
      1503609.94       941479.21      1503931.52       941517.49
      1503918.76       941844.18      1504132.66       942112.57
      1504120.39       942288.25
#Sta/Elev= 30
  4537.3  953.99  4563.4  939.19  4580.2  931.44  4607.2  920.78  4638.1  912.15
  4667.4  909.16  4711.3  907.08  4830.8  906.26  4879.2  910.53  4963.0  908.81
  4963.3  908.33  4966.1  894.56  4966.9  894.56  4969.4  889.56  5047.3  889.56
  5049.3  894.56  5051.3  899.26  5074.0  907.86  5125.7  909.39  5213.9  910.06
  5334.8  911.28  5355.1  912.14  5378.4  914.54  5417.5  917.15  5465.3  926.75
  5542.9  948.06  5558.4  951.69  5572.7  953.32  5601.4  954.77  5707.4  964.05
#Mann=6,-1,0
  4537.3    0.14       0  4966.9    0.04       0  5049.3    0.14       0
  5213.9    0.08       0  5378.4    0.14       0  5542.9    0.08       0
Bank Sta=4966.9,5049.3
XS Rating Curve= 0
Exp/Cntr=0.3,0.1

Type RM Length L Ch R = 1,36008,493,493,493
BEGIN DESCRIPTION:
Fisher River 72.0
END DESCRIPTION:
XS GIS Cut Line= 3
      1503609.90       941962.85      1503854.95       942041.99
      1504094.89       942289.58
#Sta/Elev= 30
  4857.2  953.05  4884.3  941.22  4929.8  910.31  4947.5  903.21  4956.9  894.51
  4959.4  889.51  5044.5  889.51  5047.6  894.51  5049.8  894.51  5050.8  896.89
  5055.3  899.61  5061.4  904.34  5064.7  906.02  5087.5  909.08  5132.4  910.96
  5150.6  910.03  5159.3  910.63  5170.7  910.07  5211.4  911.88  5231.4  913.30
  5245.2  915.71  5253.6  918.74  5274.1  926.13  5289.6  931.16  5323.4  943.69
  5356.6  953.26  5368.6  956.22  5411.9  959.43  5442.1  962.87  5459.5  964.27
#Mann=6,-1,0
  4857.2    0.14       0  4956.9    0.04       0  5047.6    0.14       0
  5150.6    0.08       0  5253.6    0.14       0  5356.6    0.08       0
Bank Sta=4956.9,5047.6
XS Rating Curve= 0
Exp/Cntr=0.3,0.1

Type RM Length L Ch R = 1,35515,505,505,505
BEGIN DESCRIPTION:
Fisher River 71.0
END DESCRIPTION:
XS GIS Cut Line= 3
      1503431.25       942225.71      1503479.76       942330.40
      1503630.33       942626.42
#Sta/Elev= 30
  4751.5  941.07  4756.3  940.06  4771.9  935.65  4785.6  931.07  4789.5  929.95
  4806.7  923.87  4815.1  920.08  4832.0  915.53  4839.6  913.03  4864.3  908.96
  4879.6  907.72  4906.2  906.44  4918.4  906.15  4931.0  906.15  4940.6  902.74
  4950.1  900.52  4956.9  894.46  4959.4  889.46  5047.0  889.46  5050.0  894.46
  5051.1  894.46  5053.9  900.26  5062.2  905.23  5092.2  915.05  5098.3  917.34
  5107.2  921.39  5148.6  942.52  5155.5  945.30  5185.7  964.62  5199.0  968.84
#Mann=3,-1,0
  4751.5    0.14       0  4956.9    0.04       0  5050.0    0.14       0
Bank Sta=4956.9,5050
XS Rating Curve= 0
Exp/Cntr=0.3,0.1

Type RM Length L Ch R = 1,35010,502,502,502
BEGIN DESCRIPTION:
Fisher River 70.0
END DESCRIPTION:
XS GIS Cut Line= 3
      1503298.58       942223.18      1503076.50       942391.65
      1502999.94       942583.05
#Sta/Elev= 30
  4674.3  935.68  4691.5  933.88  4709.6  931.40  4728.8  927.29  4749.8  924.17
  4793.1  914.37  4807.6  911.87  4821.6  910.96  4837.4  909.10  4884.1  908.87
  4902.3  906.96  4922.3  906.02  4953.1  899.54  4956.9  894.41  4959.4  889.41
  5040.6  889.41  5041.1  894.41  5044.4  896.55  5046.7  897.54  5052.3  902.20
  5066.0  905.25  5074.7  911.22  5091.3  920.23  5102.9  929.69  5103.8  931.08
  5112.9  939.66  5121.0  952.22  5136.2  958.71  5149.1  965.16  5159.2  970.86
#Mann=3,-1,0
  4674.3    0.14       0  4956.9    0.04       0  5041.1    0.14       0
Bank Sta=4956.9,5041.1
XS Rating Curve= 0
Exp/Cntr=0.3,0.1

Type RM Length L Ch R = 1,34508,519,519,519
BEGIN DESCRIPTION:
Fisher River 69.0
END DESCRIPTION:
XS GIS Cut Line= 3
      1502563.49       942136.44      1502589.01       942526.92
      1502739.62       942588.19
#Sta/Elev= 30
  4816.2  960.59  4825.9  957.19  4860.3  941.48  4888.3  930.75  4912.1  918.54
  4919.2  914.15  4924.2  912.44  4929.4  909.00  4939.7  904.45  4956.9  892.08
  4959.4  887.08  5045.5  887.08  5046.4  892.08  5047.3  892.08  5047.7  893.77
  5059.5  898.35  5062.2  900.23  5078.8  905.55  5130.4  907.04  5143.2  913.62
  5155.7  921.47  5172.8  927.75  5207.5  937.49  5227.6  941.54  5235.9  942.42
  5252.7  946.40  5271.6  948.40  5310.6  955.33  5338.5  961.37  5370.1  966.24
#Mann=3,-1,0
  4816.2    0.14       0  4956.9    0.04       0  5046.4    0.14       0
Bank Sta=4956.9,5046.4
XS Rating Curve= 0
Exp/Cntr=0.3,0.1

Type RM Length L Ch R = 1,33989,495,495,495
BEGIN DESCRIPTION:
Fisher River 68.0
END DESCRIPTION:
XS GIS Cut Line= 3
      1501975.00       942275.00      1502147.46       942598.39
      1502229.13       942782.15
#Sta/Elev= 30
  4749.1  962.49  4770.0  959.20  4789.3  955.28  4809.1  951.99  4828.1  946.70
  4838.8  942.75  4855.5  937.50  4898.2  922.26  4917.5  913.04  4931.5  905.52
  4960.6  892.65  4961.1  890.65  4963.0  885.65  5040.6  885.65  5043.1  890.65
  5057.1  898.17  5113.4  905.44  5128.5  905.52  5142.3  906.87  5153.1  910.05
  5173.1  920.89  5183.8  925.15  5202.9  934.10  5216.3  940.72  5230.9  949.50
  5240.1  952.71  5243.7  954.98  5260.3  960.25  5277.5  964.64  5316.7  969.64
#Mann=3,-1,0
  4749.1    0.14       0  4961.1    0.04       0  5043.1    0.14       0
Bank Sta=4961.1,5043.1
XS Rating Curve= 0
Exp/Cntr=0.3,0.1

Type RM Length L Ch R = 1,33494,494,494,494
BEGIN DESCRIPTION:
Fisher River 67.0
END DESCRIPTION:
XS GIS Cut Line= 4
      1501759.51       942348.26      1501693.15       942626.46
      1501652.32       942784.70      1501468.57       942953.14
#Sta/Elev= 30
  4614.2  948.18  4674.3  941.24  4715.3  933.73  4735.4  928.71  4754.1  925.27
  4779.6  916.97  4805.0  906.78  4822.1  903.24  4847.8  903.91  4912.4  903.38
  4926.6  904.50  4944.6  903.44  4955.2  903.79  4955.7  903.19  4956.5  889.89
  4956.6  884.89  5047.1  884.89  5047.2  889.89  5048.5  897.56  5050.0  898.67
  5069.5  905.58  5075.4  906.95  5099.1  907.71  5129.2  910.82  5157.4  917.81
  5230.1  947.52  5235.3  948.84  5257.4  959.26  5288.1  971.90  5312.9  980.22
#Mann=3,-1,0
  4614.2    0.14       0  4956.5    0.04       0  5047.2    0.14       0
Bank Sta=4956.5,5047.2
XS Rating Curve= 0
Exp/Cntr=0.3,0.1

Type RM Length L Ch R = 1,33000,492,492,492
BEGIN DESCRIPTION:
Fisher River 66.0
END DESCRIPTION:
XS GIS Cut Line= 3
      1501716.12       942287.01      1501527.25       942299.77
      1501213.28       942325.29
#Sta/Elev= 30
  4731.8  941.23  4761.6  935.16  4809.4  922.89  4828.4  918.70  4834.5  917.01
  4850.8  911.43  4859.1  909.56  4872.5  907.36  4898.6  906.82  4915.1  904.74
  4920.8  903.42  4951.3  900.28  4954.2  899.51  4961.8  889.32  4965.2  884.32
  5029.9  884.32  5035.1  889.32  5051.5  896.95  5076.5  907.77  5103.7  923.37
  5105.9  924.27  5117.7  931.94  5141.5  946.69  5157.0  955.08  5163.7  958.33
  5183.9  969.47  5192.1  973.09  5204.0  977.54  5216.3  980.71  5236.1  983.65
#Mann=3,-1,0
  4731.8    0.14       0  4961.8    0.04       0  5035.1    0.14       0
Bank Sta=4961.8,5035.1
XS Rating Curve= 0
Exp/Cntr=0.3,0.1

Type RM Length L Ch R = 1,32508,515,515,515
BEGIN DESCRIPTION:
Fisher River 65.0
END DESCRIPTION:
XS GIS Cut Line= 4
      1501807.98       941848.01      1501665.08       941850.56
      1501358.80       941789.31      1501272.03       941944.99
#Sta/Elev= 30
  4723.9  948.11  4757.2  941.80  4822.5  927.09  4898.7  904.43  4930.3  904.05
  4941.2  902.01  4958.9  896.03  4963.8  892.12  4964.7  888.73  4966.9  883.73
  5036.4  883.73  5037.4  888.73  5039.3  892.31  5048.9  898.71  5054.5  899.55
  5074.7  899.63  5095.7  900.85  5117.2  902.89  5128.4  905.57  5140.3  909.25
  5143.7  909.93  5164.7  917.97  5185.3  922.55  5209.7  924.65  5217.0  925.69
  5240.9  930.56  5270.0  933.92  5334.8  944.79  5349.8  945.23  5357.4  946.74
#Mann=3,-1,0
  4723.9    0.14       0  4964.7    0.04       0  5037.4    0.14       0
Bank Sta=4964.7,5037.4
XS Rating Curve= 0
Exp/Cntr=0.3,0.1

Type RM Length L Ch R = 1,31993,495,495,495
BEGIN DESCRIPTION:
Fisher River 64.0
END DESCRIPTION:
XS GIS Cut Line= 3
      1501966.20       941460.05      1501864.16       941439.64
      1501525.03       941225.02
#Sta/Elev= 30
  4713.8  967.09  4727.2  962.62  4734.1  960.60  4758.1  950.99  4767.8  946.86
  4774.9  944.48  4787.6  938.38  4828.4  920.07  4833.7  917.26  4853.9  907.41
  4867.7  904.18  4883.6  903.54  4889.2  902.97  4892.8  902.18  4909.7  901.67
  4946.6  895.09  4950.9  894.49  4955.4  887.74  4956.5  882.74  5041.5  882.74
  5043.6  887.74  5045.5  890.26  5088.5  906.42  5090.8  905.58  5101.0  910.01
  5108.2  914.01  5141.9  927.66  5170.9  938.51  5181.8  942.03  5219.2  950.51
#Mann=3,-1,0
  4713.8    0.14       0  4955.4    0.04       0  5043.6    0.14       0
Bank Sta=4955.4,5043.6
XS Rating Curve= 0
Exp/Cntr=0.3,0.1

Type RM Length L Ch R = 1,31498,495,495,495
BEGIN DESCRIPTION:
Fisher River 63.0
END DESCRIPTION:
XS GIS Cut Line= 3
      1502017.29       940870.48      1501915.20       940873.03
      1501542.59       941013.40
#Sta/Elev= 30
  4805.4  981.80  4808.9  981.04  4815.8  977.00  4820.7  977.09  4837.6  967.22
  4844.6  958.59  4850.8  955.31  4862.0  946.65  4883.7  927.98  4896.8  918.70
  4900.5  917.02  4930.3  908.51  4947.4  888.15  4950.3  887.62  4950.9  886.21
  4953.4  881.21  5040.4  881.21  5041.2  886.21  5041.5  886.21  5041.8  889.72
  5042.4  892.84  5051.7  895.08  5090.8  897.65  5115.0  901.67  5147.5  908.32
  5161.3  909.55  5186.2  914.37  5233.4  920.90  5280.1  928.86  5305.7  930.92
#Mann=3,-1,0
  4805.4    0.14       0  4950.9    0.04       0  5041.2    0.14       0
Bank Sta=4950.9,5041.2
XS Rating Curve= 0
Exp/Cntr=0.3,0.1

Type RM Length L Ch R = 1,31003,526,526,526
BEGIN DESCRIPTION:
Fisher River 62.0
END DESCRIPTION:
XS GIS Cut Line= 3
      1501762.07       940296.21      1501695.70       940395.75
      1501399.61       940717.37
#Sta/Elev= 30
  4782.9  948.09  4809.3  940.09  4827.7  935.15  4847.5  930.26  4879.2  925.47
  4898.5  919.19  4910.5  913.61  4917.2  911.05  4919.4  908.36  4936.6  898.02
  4948.7  884.78  4950.7  884.78  4951.4  879.78  5027.5  879.78  5029.4  884.78
  5033.5  888.48  5037.9  890.76  5067.4  894.70  5087.1  896.29  5092.3  896.35
  5101.1  896.65  5134.4  900.92  5146.9  902.24  5158.6  904.44  5166.7  907.36
  5207.1  920.46  5249.5  931.80  5277.9  939.22  5325.6  949.99  5339.7  952.48
#Mann=4,-1,0
  4782.9    0.14       0  4950.7    0.04       0  5029.4    0.08       0
  5092.3    0.14       0
Bank Sta=4950.7,5029.4
XS Rating Curve= 0
Exp/Cntr=0.3,0.1

Type RM Length L Ch R = 1,30477,463,463,463
BEGIN DESCRIPTION:
Fisher River 61.0
END DESCRIPTION:
XS GIS Cut Line= 4
      1501375.01       939974.98      1501276.39       940078.33
      1501187.80       940171.15      1500983.59       940252.83
#Sta/Elev= 30
  4796.8  965.24  4812.9  958.00  4823.8  949.96  4833.7  946.67  4843.8  940.72
  4853.5  931.14  4872.5  919.02  4891.8  911.00  4904.1  904.37  4908.9  903.01
  4924.7  894.60  4926.7  892.96  4935.5  892.69  4953.4  889.76  4958.0  883.75
  4960.0  878.75  5039.3  878.75  5042.1  883.75  5044.6  886.91  5046.3  888.21
  5055.5  892.61  5062.6  893.97  5068.3  894.16  5076.1  893.28  5092.0  893.77
  5124.3  897.20  5193.9  915.69  5220.8  921.82  5255.0  931.83  5287.9  940.13
#Mann=3,-1,0
  4796.8    0.14       0  4958.0    0.04       0  5042.1    0.14       0
Bank Sta=4958,5042.1
XS Rating Curve= 0
Exp/Cntr=0.3,0.1

Type RM Length L Ch R = 1,30014,579,579,579
BEGIN DESCRIPTION:
Fisher River 60.0
END DESCRIPTION:
XS GIS Cut Line= 5
      1501366.44       939729.60      1501072.94       939693.87
      1500917.25       939767.89      1500850.89       939875.08
      1500820.27       940025.67
#Sta/Elev= 30
  4603.8  976.88  4627.7  972.26  4654.0  966.23  4723.4  944.63  4764.6  930.87
  4819.2  907.05  4822.6  906.51  4840.1  901.37  4856.0  898.95  4889.6  897.75
  4899.5  894.97  4909.6  890.91  4947.6  882.99  4952.7  882.99  4954.9  877.99
  5044.6  877.99  5046.9  882.99  5053.6  883.02  5053.7  885.70  5058.7  888.35
  5065.5  888.14  5096.9  894.19  5115.2  896.03  5159.3  908.50  5188.9  915.04
  5252.1  923.20  5266.2  924.44  5311.6  930.98  5332.7  937.04  5351.6  939.80
#Mann=3,-1,0
  4603.8    0.14       0  4952.7    0.04       0  5046.9    0.14       0
Bank Sta=4952.7,5046.9
XS Rating Curve= 0
Exp/Cntr=0.3,0.1

Type RM Length L Ch R = 1,29435,506,506,506
BEGIN DESCRIPTION:
Fisher River 59.0
END DESCRIPTION:
XS GIS Cut Line= 3
      1501409.80       939328.88      1500896.83       939150.23
      1500728.43       939140.02
#Sta/Elev= 30
  4518.5  959.35  4583.7  948.57  4611.4  940.51  4665.1  916.26  4683.6  909.84
  4727.2  899.24  4754.8  897.29  4846.4  899.66  4916.5  897.50  4937.8  891.92
  4940.3  888.54  4942.0  881.84  4942.9  881.84  4945.3  876.84  5050.9  876.84
  5051.0  881.84  5051.4  881.87  5052.2  887.78  5056.3  891.05  5064.4  892.60
  5078.4  899.86  5106.2  920.32  5148.6  945.27  5159.0  952.80  5169.8  965.71
  5172.0  967.15  5180.6  970.86  5202.4  983.77  5221.4  990.26  5230.4  991.95
#Mann=3,-1,0
  4518.5    0.14       0  4942.9    0.04       0  5051.0    0.14       0
Bank Sta=4942.9,5051
XS Rating Curve= 0
Exp/Cntr=0.3,0.1

Type RM Length L Ch R = 1,28929,492,492,492
BEGIN DESCRIPTION:
Fisher River 58.0
END DESCRIPTION:
XS GIS Cut Line= 4
      1501445.59       938609.14      1501190.35       938698.47
      1500965.75       938670.40      1500840.72       938723.98
#Sta/Elev= 30
  4643.7  937.12  4663.6  932.73  4697.6  923.83  4725.9  918.65  4750.6  913.33
  4765.4  910.78  4791.0  904.38  4843.5  898.84  4867.7  895.87  4901.2  894.69
  4921.6  893.35  4926.7  893.39  4928.9  892.94  4931.1  880.83  4934.3  875.83
  5051.4  875.83  5055.7  880.83  5056.8  880.84  5057.2  882.43  5063.0  891.35
  5077.3  892.01  5118.0  897.88  5138.8  899.93  5146.2  901.10  5162.3  902.82
  5175.3  908.60  5193.7  915.98  5223.2  926.44  5240.8  931.46  5276.5  942.41
#Mann=3,-1,0
  4643.7    0.14       0  4931.1    0.04       0  5055.7    0.14       0
Bank Sta=4931.1,5055.7
XS Rating Curve= 0
Exp/Cntr=0.3,0.1

Type RM Length L Ch R = 1,28437,439,439,439
BEGIN DESCRIPTION:
Fisher River 57.0
END DESCRIPTION:
XS GIS Cut Line= 4
      1501402.21       938129.29      1501274.58       938205.88
      1501146.96       938213.54      1500963.16       938325.86
#Sta/Elev= 30
  4787.5  947.88  4799.1  942.46  4808.8  940.20  4839.0  926.47  4864.3  912.08
  4882.9  904.29  4892.7  899.28  4901.0  896.27  4919.1  888.11  4935.5  881.26
  4941.7  879.13  4949.6  879.39  4954.0  879.10  4956.5  874.10  5035.6  874.10
  5036.5  879.10  5037.5  894.17  5038.4  894.02  5043.0  895.03  5061.8  890.93
  5064.2  891.54  5078.2  893.24  5083.7  894.68  5092.9  896.08  5142.9  914.75
  5148.6  916.29  5169.8  923.86  5208.4  934.03  5221.8  938.04  5279.6  949.81
#Mann=3,-1,0
  4787.5    0.14       0  4954.0    0.04       0  5036.5    0.14       0
Bank Sta=4954,5036.5
XS Rating Curve= 0
Exp/Cntr=0.3,0.1

Type RM Length L Ch R = 1,27998,502,502,502
BEGIN DESCRIPTION:
Fisher River 56.0
END DESCRIPTION:
XS GIS Cut Line= 3
      1500993.83       937787.28      1500891.73       938017.01
      1500889.18       938221.20
#Sta/Elev= 30
  4812.2  962.65  4827.8  950.11  4832.2  947.92  4850.4  939.14  4859.5  933.16
  4875.1  922.47  4898.2  909.87  4912.6  904.41  4924.3  899.26  4950.7  890.98
  4961.1  883.51  4962.4  877.42  4962.9  872.42  5045.9  872.42  5046.0  877.42
  5055.5  888.03  5060.0  891.73  5079.9  893.90  5097.8  894.82  5109.9  898.03
  5118.5  899.08  5124.8  900.01  5135.4  902.82  5181.2  920.15  5189.2  922.44
  5204.3  926.03  5208.1  926.77  5232.5  931.03  5248.2  934.82  5267.8  937.97
#Mann=3,-1,0
  4812.2    0.14       0  4962.4    0.04       0  5046.0    0.14       0
Bank Sta=4962.4,5046
XS Rating Curve= 0
Exp/Cntr=0.3,0.1

Type RM Length L Ch R = 1,27496,486,486,486
BEGIN DESCRIPTION:
Fisher River 55.0
END DESCRIPTION:
XS GIS Cut Line= 3
      1500468.04       937657.18      1500414.45       937920.02
      1500434.86       938096.09
#Sta/Elev= 30
  4819.6  940.24  4835.1  932.93  4841.4  930.86  4868.1  919.57  4899.8  904.85
  4922.8  899.38  4944.4  896.42  4949.8  893.33  4956.4  876.41  4958.9  871.41
  5037.1  871.41  5038.6  876.41  5045.7  882.88  5052.5  887.36  5065.5  889.23
  5083.8  891.17  5093.0  893.52  5098.0  894.27  5106.2  896.24  5119.1  900.23
  5123.6  901.72  5136.7  906.99  5151.6  909.78  5167.2  915.20  5187.4  920.64
  5199.0  924.34  5231.6  932.33  5245.8  934.70  5261.7  936.89  5265.1  937.62
#Mann=3,-1,0
  4819.6    0.14       0  4956.4    0.04       0  5038.6    0.14       0
Bank Sta=4956.4,5038.6
XS Rating Curve= 0
Exp/Cntr=0.3,0.1

Type RM Length L Ch R = 1,27010,510,510,510
BEGIN DESCRIPTION:
Fisher River 54.0
END DESCRIPTION:
XS GIS Cut Line= 4
      1500082.61       937618.87      1499960.14       937692.87
      1499942.27       937889.39      1499893.79       938062.92
#Sta/Elev= 30
  4710.3  929.06  4742.6  923.90  4764.4  919.18  4780.2  916.53  4802.5  911.60
  4816.3  908.24  4857.6  896.39  4875.0  893.51  4900.9  890.61  4926.2  889.71
  4949.1  876.57  4951.3  875.68  4954.8  870.68  5033.0  870.68  5033.3  875.68
  5041.1  883.91  5048.8  886.73  5076.4  889.60  5099.3  898.73  5106.9  902.32
  5110.5  904.59  5115.4  908.17  5124.0  915.25  5155.1  928.24  5166.2  935.04
  5172.9  938.56  5183.5  944.99  5190.6  948.65  5208.2  956.74  5230.9  966.57
#Mann=3,-1,0
  4710.3    0.14       0  4951.3    0.04       0  5033.3    0.14       0
Bank Sta=4951.3,5033.3
XS Rating Curve= 0
Exp/Cntr=0.3,0.1

Type RM Length L Ch R = 1,26500,499,499,499
BEGIN DESCRIPTION:
Fisher River 53.0
END DESCRIPTION:
XS GIS Cut Line= 3
      1499702.34       937396.82      1499531.66       937574.81
      1499367.98       937746.49
#Sta/Elev= 30
  4753.4  921.74  4757.9  920.80  4787.7  912.89  4810.1  907.57  4832.1  901.26
  4859.0  895.29  4877.2  894.18  4913.4  890.88  4939.0  888.98  4951.5  886.16
  4959.6  878.51  4960.2  875.32  4961.0  870.32  5036.2  870.32  5037.0  875.32
  5042.8  879.83  5058.3  888.06  5071.4  891.44  5082.9  899.15  5091.6  904.26
  5094.6  906.43  5109.0  915.30  5120.4  922.93  5130.2  930.04  5147.0  940.80
  5151.1  943.74  5188.6  965.79  5195.5  969.61  5226.0  985.35  5237.2  990.08
#Mann=3,-1,0
  4753.4    0.14       0  4960.2    0.04       0  5037.0    0.14       0
Bank Sta=4960.2,5037
XS Rating Curve= 0
Exp/Cntr=0.3,0.1

Type RM Length L Ch R = 1,26001,496,496,496
BEGIN DESCRIPTION:
Fisher River 52.0
END DESCRIPTION:
XS GIS Cut Line= 3
      1499380.74       937044.60      1499117.88       937274.29
      1498939.21       937427.44
#Sta/Elev= 30
  4776.1  936.70  4792.6  933.12  4812.5  926.95  4830.2  922.58  4848.0  916.31
  4884.0  904.99  4902.7  898.62  4918.8  892.09  4938.6  887.55  4958.7  879.23
  4962.7  875.29  4965.8  870.29  5039.7  870.29  5041.8  875.29  5042.6  881.20
  5045.3  883.60  5059.3  883.62  5108.3  888.56  5135.3  888.96  5152.6  889.42
  5168.9  892.23  5185.0  895.89  5201.9  901.15  5213.2  905.48  5217.7  907.19
  5253.6  924.92  5279.4  938.27  5326.2  967.14  5354.3  978.73  5360.5  980.65
#Mann=5,-1,0
  4776.1    0.14       0  4962.7    0.04       0  5041.8    0.14       0
  5135.3    0.08       0  5213.2    0.14       0
Bank Sta=4962.7,5041.8
XS Rating Curve= 0
Exp/Cntr=0.3,0.1

Type RM Length L Ch R = 1,25505,493,493,493
BEGIN DESCRIPTION:
Fisher River 51.0
END DESCRIPTION:
XS GIS Cut Line= 3
      1499411.36       936924.60      1498951.98       936679.60
      1498949.43       936546.85
#Sta/Elev= 30
  4621.5  941.86  4666.1  934.66  4697.7  927.27  4724.6  922.10  4823.3  897.26
  4847.5  893.35  4874.0  891.27  4887.4  891.38  4903.1  889.27  4930.0  887.71
  4949.8  878.29  4954.0  875.25  4956.5  870.25  5039.8  870.25  5039.9  875.25
  5042.0  875.25  5043.4  878.07  5052.6  887.70  5070.0  897.52  5078.6  903.98
  5093.5  912.03  5121.4  933.71  5133.5  937.19  5142.1  937.89  5152.0  940.59
  5167.7  946.79  5181.8  949.12  5200.5  954.09  5256.7  964.36  5274.9  966.32
#Mann=3,-1,0
  4621.5    0.14       0  4954.0    0.04       0  5039.9    0.14       0
Bank Sta=4954,5039.9
XS Rating Curve= 0
Exp/Cntr=0.3,0.1

Type RM Length L Ch R = 1,25012,512,512,512
BEGIN DESCRIPTION:
Fisher River 50.0
END DESCRIPTION:
XS GIS Cut Line= 3
      1499635.98       936712.76      1499544.12       936559.64
      1499296.53       936217.61
#Sta/Elev= 30
  4664.0  937.75  4742.2  921.13  4755.8  920.24  4797.3  909.52  4847.0  894.99
  4850.8  893.40  4865.1  888.93  4870.8  886.25  4884.4  883.44  4902.0  887.59
  4908.5  887.59  4912.9  888.20  4922.9  886.64  4937.5  886.48  4944.6  884.41
  4954.0  873.99  4954.1  868.99  5045.1  868.99  5046.0  873.99  5052.3  880.31
  5063.4  892.65  5080.3  902.44  5085.2  906.36  5112.4  925.55  5137.1  944.37
  5155.5  954.72  5169.9  963.66  5214.7  981.99  5245.9  989.27  5264.8  992.02
#Mann=3,-1,0
  4664.0    0.14       0  4954.0    0.04       0  5046.0    0.14       0
Bank Sta=4954,5046
XS Rating Curve= 0
Exp/Cntr=0.3,0.1

Type RM Length L Ch R = 1,24500,493,493,493
BEGIN DESCRIPTION:
Fisher River 49.0
END DESCRIPTION:
XS GIS Cut Line= 3
      1500031.60       936444.78      1499978.01       936268.68
      1499727.87       935959.84
#Sta/Elev= 30
  4638.9  964.70  4693.6  946.04  4706.7  945.75  4718.0  944.20  4753.6  923.22
  4760.7  920.33  4837.9  894.38  4849.8  891.10  4870.8  887.20  4936.1  885.69
  4948.7  882.36  4951.9  877.85  4955.5  873.89  4955.6  873.13  4956.4  873.13
  4956.5  868.13  5051.2  868.13  5051.3  873.13  5058.2  879.21  5060.6  882.81
  5087.4  893.52  5107.6  907.60  5118.6  914.18  5128.3  923.84  5139.1  929.29
  5150.8  936.73  5160.6  940.77  5182.1  948.04  5212.5  955.13  5220.4  955.57
#Mann=3,-1,0
  4638.9    0.14       0  4956.4    0.04       0  5051.3    0.14       0
Bank Sta=4956.4,5051.3
XS Rating Curve= 0
Exp/Cntr=0.3,0.1

Type RM Length L Ch R = 1,24007,507,507,507
BEGIN DESCRIPTION:
Fisher River 48.0
END DESCRIPTION:
XS GIS Cut Line= 3
      1500394.05       935842.46      1500008.63       935694.42
      1499863.11       935709.73
#Sta/Elev= 30
  4769.4  987.34  4799.4  968.45  4809.8  963.04  4820.4  954.38  4883.6  915.74
  4893.4  908.98  4914.4  896.62  4925.6  890.46  4941.9  883.55  4946.7  880.52
  4955.8  878.49  4957.5  872.26  4957.6  867.55  5044.3  867.55  5044.4  872.55
  5045.6  876.33  5052.0  880.82  5061.7  885.32  5086.2  885.42  5099.5  884.17
  5107.5  885.92  5127.7  886.47  5147.7  889.59  5158.5  890.15  5168.9  894.38
  5201.0  903.24  5225.1  908.73  5245.3  914.77  5271.7  918.57  5328.6  930.05
#Mann=3,-1,0
  4769.4    0.14       0  4957.5    0.04       0  5044.4    0.14       0
Bank Sta=4957.5,5044.4
XS Rating Curve= 0
Exp/Cntr=0.3,0.1

Type RM Length L Ch R = 1,23500,489,489,489
BEGIN DESCRIPTION:
Fisher River 47.0
END DESCRIPTION:
XS GIS Cut Line= 3
      1500276.64       935199.26      1500125.63       935277.12
      1499814.64       935439.20
#Sta/Elev= 30
  4830.1  952.76  4836.1  949.35  4856.1  936.65  4880.6  922.43  4906.1  906.48
  4915.7  899.85  4923.0  895.29  4949.2  880.64  4953.6  879.03  4957.3  875.86
  4957.5  871.73  4960.4  866.73  5048.2  866.73  5049.1  871.73  5052.8  876.72
  5060.1  881.68  5065.5  884.44  5083.4  885.94  5103.1  886.34  5124.6  888.01
  5139.0  888.53  5162.7  890.90  5182.6  895.45  5197.5  897.76  5232.8  905.07
  5288.2  912.99  5315.3  917.39  5329.5  919.29  5343.5  920.00  5350.7  921.26
#Mann=3,-1,0
  4830.1    0.14       0  4957.5    0.04       0  5049.1    0.14       0
Bank Sta=4957.5,5049.1
XS Rating Curve= 0
Exp/Cntr=0.3,0.1

Type RM Length L Ch R = 1,23011,508,508,508
BEGIN DESCRIPTION:
Fisher River 46.0
END DESCRIPTION:
XS GIS Cut Line= 3
      1500100.47       934810.05      1499750.85       934871.30
      1499600.24       934912.14
#Sta/Elev= 30
  4799.8  947.66  4806.6  946.48  4817.4  946.36  4818.8  945.83  4847.7  920.58
  4853.5  917.21  4873.7  903.85  4886.5  900.73  4899.6  895.67  4911.1  891.69
  4912.3  891.73  4913.5  890.85  4915.1  886.51  4931.3  870.87  4943.8  870.52
  4948.4  869.58  4950.4  864.58  5051.0  864.58  5053.6  869.58  5055.8  877.66
  5056.5  878.44  5068.7  883.98  5129.7  885.65  5141.7  886.91  5156.5  891.95
  5163.4  893.46  5175.2  897.46  5212.4  907.48  5239.6  913.95  5310.8  927.05
#Mann=3,-1,0
  4799.8    0.14       0  4948.4    0.04       0  5053.6    0.14       0
Bank Sta=4948.4,5053.6
XS Rating Curve= 0
Exp/Cntr=0.3,0.1

Type RM Length L Ch R = 1,22503,488,488,488
BEGIN DESCRIPTION:
Fisher River 45.0
END DESCRIPTION:
XS GIS Cut Line= 3
      1500156.71       934457.84      1499847.84       934320.00
      1499661.49       934340.42
#Sta/Elev= 30
  4728.3  909.66  4746.7  907.24  4753.3  906.75  4774.6  899.80  4809.3  890.07
  4838.3  880.67  4845.0  879.40  4854.1  878.60  4876.8  878.68  4890.3  880.27
  4895.4  882.74  4901.4  881.16  4904.3  881.38  4915.7  880.55  4923.0  880.56
  4932.5  875.63  4935.3  866.96  4936.2  861.96  5048.6  861.96  5048.7  866.96
  5052.4  866.96  5053.3  869.20  5061.9  879.44  5091.1  883.27  5117.8  892.18
  5139.8  901.69  5152.4  907.71  5172.6  918.27  5218.2  942.76  5254.0  960.49
#Mann=3,-1,0
  4728.3    0.14       0  4935.3    0.04       0  5048.7    0.14       0
Bank Sta=4935.3,5048.7
XS Rating Curve= 0
Exp/Cntr=0.3,0.1

Type RM Length L Ch R = 1,22015,510,510,510
BEGIN DESCRIPTION:
Fisher River 44.0
END DESCRIPTION:
XS GIS Cut Line= 3
      1500376.13       934148.96      1500108.17       933881.01
      1499926.94       933837.61
#Sta/Elev= 30
  4686.4  909.83  4720.5  905.45  4750.5  897.40  4763.2  894.37  4795.6  887.61
  4805.6  886.46  4811.8  885.25  4851.0  883.22  4873.1  880.43  4883.9  879.92
  4890.9  878.96  4909.0  878.59  4923.0  876.27  4928.5  876.61  4937.6  878.25
  4954.8  873.35  4961.7  865.48  4963.8  860.48  5052.9  860.48  5053.8  865.48
  5065.3  869.11  5150.4  899.62  5164.8  902.96  5202.9  916.06  5205.7  917.49
  5212.7  920.01  5220.1  922.09  5229.4  925.38  5247.3  932.95  5251.7  934.34
#Mann=3,-1,0
  4686.4    0.14       0  4961.7    0.04       0  5053.8    0.14       0
Bank Sta=4961.7,5053.8
XS Rating Curve= 0
Exp/Cntr=0.3,0.1

Type RM Length L Ch R = 1,21505,510,510,510
BEGIN DESCRIPTION:
Fisher River 43.0
END DESCRIPTION:
XS GIS Cut Line= 4
      1500641.61       933944.82      1500628.84       933669.17
      1500450.18       933528.79      1500294.49       933490.50
#Sta/Elev= 30
  4619.5  905.27  4680.8  897.93  4703.6  896.55  4791.3  886.90  4821.4  884.49
  4854.0  882.70  4876.8  882.57  4888.0  883.41  4897.2  883.17  4931.6  880.36
  4939.8  879.36  4953.5  872.89  4958.0  869.34  4959.1  865.45  4961.3  860.45
  5056.5  860.45  5058.7  865.45  5059.8  865.45  5068.3  878.12  5126.8  883.52
  5154.4  891.49  5183.7  904.01  5198.2  912.47  5208.1  916.76  5230.9  929.18
  5247.7  936.30  5253.9  937.80  5269.0  943.44  5276.4  946.97  5283.0  949.20
#Mann=3,-1,0
  4619.5    0.14       0  4959.1    0.04       0  5058.7    0.14       0
Bank Sta=4959.1,5058.7
XS Rating Curve= 0
Exp/Cntr=0.3,0.1

Type RM Length L Ch R = 1,20995,488,488,488
BEGIN DESCRIPTION:
Fisher River 42.0
END DESCRIPTION:
XS GIS Cut Line= 4
      1500965.77       933082.12      1500848.34       933151.05
      1500705.41       933171.47      1500434.82       933225.07
#Sta/Elev= 30
  4791.0  953.17  4808.5  950.39  4823.1  945.26  4839.0  938.44  4857.3  928.26
  4877.5  911.70  4885.5  906.17  4887.8  905.43  4899.8  893.95  4927.2  885.64
  4942.9  882.06  4954.2  865.11  4955.8  860.11  5045.8  860.11  5045.9  865.11
  5048.4  873.99  5048.7  874.37  5061.8  876.85  5073.7  877.01  5137.9  882.17
  5161.9  885.88  5224.9  899.59  5237.2  901.46  5252.1  902.95  5263.1  905.10
  5272.8  907.96  5295.5  909.28  5313.0  911.43  5328.7  912.68  5347.4  913.57
#Mann=3,-1,0
  4791.0    0.14       0  4954.2    0.04       0  5045.9    0.08       0
Bank Sta=4954.2,5045.9
XS Rating Curve= 0
Exp/Cntr=0.3,0.1

Type RM Length L Ch R = 1,20507,497,497,497
BEGIN DESCRIPTION:
Fisher River 41.0
END DESCRIPTION:
XS GIS Cut Line= 4
      1500779.41       932668.67      1500725.83       932696.74
      1500530.06       932718.80      1500320.03       932913.67
#Sta/Elev= 30
  4821.0  916.12  4836.1  918.90  4839.8  918.60  4845.1  917.97  4856.5  913.46
  4860.2  912.73  4880.2  900.69  4880.4  900.45  4939.7  869.93  4951.6  864.75
  4953.3  864.19  4955.8  859.19  5050.8  859.19  5051.5  864.19  5053.1  864.24
  5055.8  867.62  5058.0  870.68  5065.5  878.70  5076.3  878.99  5107.7  880.90
  5126.1  882.23  5175.9  886.69  5193.8  889.43  5210.2  891.59  5225.9  894.08
  5234.6  894.42  5283.5  900.39  5324.1  903.72  5333.4  904.77  5365.0  906.65
#Mann=4,-1,0
  4821.0    0.14       0  4953.3    0.04       0  5051.5    0.14       0
  5107.7    0.08       0
Bank Sta=4953.3,5051.5
XS Rating Curve= 0
Exp/Cntr=0.3,0.1

Type RM Length L Ch R = 1,20010,518,518,518
BEGIN DESCRIPTION:
Fisher River 40.0
END DESCRIPTION:
XS GIS Cut Line= 3
      1500774.33       932285.82      1500667.13       932211.80
      1500161.74       932227.12
#Sta/Elev= 30
  4779.0  902.93  4804.7  900.15  4852.4  885.18  4882.7  880.05  4894.0  876.38
  4901.4  873.52  4948.6  864.43  4953.3  862.89  4955.8  857.89  5042.2  857.89
  5042.3  862.89  5042.8  869.42  5045.0  874.48  5051.0  875.82  5055.1  876.25
  5059.0  877.30  5066.1  878.24  5087.8  878.84  5091.9  879.27  5135.5  879.62
  5181.2  882.16  5200.4  883.63  5228.6  890.27  5234.5  891.69  5256.9  894.38
  5281.0  895.90  5321.8  899.71  5371.7  902.24  5393.9  902.78  5414.9  902.50
#Mann=6,-1,0
  4779.0    0.14       0  4953.3    0.04       0  5042.3    0.14       0
  5135.5    0.08       0  5228.6    0.14       0  5321.8    0.08       0
Bank Sta=4953.3,5042.3
XS Rating Curve= 0
Exp/Cntr=0.3,0.1

Type RM Length L Ch R = 1,19492,503,503,503
BEGIN DESCRIPTION:
Fisher River 39.0
END DESCRIPTION:
XS GIS Cut Line= 3
      1500498.65       931612.04      1500312.36       931846.82
      1500146.48       932119.88
#Sta/Elev= 30
  4797.6  971.12  4826.1  970.12  4843.8  960.53  4853.1  958.47  4861.8  953.22
  4893.3  924.98  4907.5  918.71  4924.7  913.44  4927.9  910.41  4938.1  892.34
  4953.3  861.87  4953.4  856.87  5044.5  856.87  5044.6  861.87  5049.7  874.48
  5054.8  874.18  5069.0  877.32  5093.7  876.74  5099.2  877.12  5132.3  877.21
  5162.9  878.66  5189.2  880.68  5216.6  886.73  5225.2  887.98  5248.8  892.94
  5259.3  894.57  5297.4  895.98  5324.3  897.76  5376.4  901.19  5416.8  902.44
#Mann=6,-1,0
  4797.6    0.14       0  4953.3    0.04       0  5044.6    0.14       0
  5132.3    0.08       0  5225.2    0.14       0  5324.3    0.08       0
Bank Sta=4953.3,5044.6
XS Rating Curve= 0
Exp/Cntr=0.3,0.1

Type RM Length L Ch R = 1,18989,474,474,474
BEGIN DESCRIPTION:
Fisher River 38.0
END DESCRIPTION:
XS GIS Cut Line= 3
      1500164.36       931461.42      1499995.87       931469.08
      1499710.05       931793.19
#Sta/Elev= 30
  4722.2  929.83  4732.6  929.47  4749.6  927.61  4767.1  924.70  4781.6  921.84
  4794.2  919.84  4808.5  916.28  4826.2  913.54  4851.7  906.65  4857.1  905.64
  4866.9  904.93  4889.2  901.41  4890.9  899.00  4900.6  889.00  4904.8  887.73
  4930.2  874.84  4944.6  861.57  4949.6  856.57  5045.7  856.57  5045.8  861.57
  5048.4  867.21  5055.1  876.69  5070.5  875.70  5105.0  876.68  5130.0  877.99
  5169.8  880.51  5198.8  883.24  5275.8  895.30  5289.5  896.79  5323.0  897.26
#Mann=4,-1,0
  4722.2    0.14       0  4944.6    0.04       0  5045.8    0.14       0
  5130.0    0.08       0
Bank Sta=4944.6,5045.8
XS Rating Curve= 0
Exp/Cntr=0.3,0.1

Type RM Length L Ch R = 1,18515,303,303,303
BEGIN DESCRIPTION:
Fisher River 37.0
END DESCRIPTION:
XS GIS Cut Line= 4
      1500192.43       931047.95      1499886.12       931060.71
      1499600.27       931185.78      1499444.56       931341.49
#Sta/Elev= 30
  4496.7  909.04  4503.8  908.78  4558.1  899.11  4585.6  894.82  4641.9  889.38
  4703.5  886.55  4757.3  889.64  4776.3  892.79  4795.8  893.73  4839.8  892.46
  4888.5  886.71  4900.8  886.42  4919.3  880.13  4931.2  874.19  4952.3  871.54
  4954.2  861.29  4955.1  856.29  5050.5  856.29  5053.4  861.29  5059.4  871.05
  5061.4  873.21  5105.5  873.59  5140.5  876.78  5166.7  877.31  5191.0  881.66
  5213.3  891.68  5231.7  902.79  5249.1  910.01  5318.4  932.69  5335.5  934.23
#Mann=4,-1,0
  4496.7    0.08       0  4558.1    0.14       0  4954.2    0.04       0
  5053.4    0.08       0
Bank Sta=4954.2,5053.4
XS Rating Curve= 0
Exp/Cntr=0.5,0.3
