--- Forbush Creek.prj (project) ---

Proj Title=Forbush Creek Limited Detail Study
Current Plan=p01
Default Exp/Contr=0.3,0.1
English Units
Geom File=g01
Flow File=f01
Plan File=p01
Y Axis Title=Elevation
X Axis Title(PF)=Main Channel Distance
X Axis Title(XS)=Station
BEGIN DESCRIPTION:
Forbush Creek
END DESCRIPTION:
DSS Export Rating Curves= 0
DSS Export Rating Curve Sorted= 0
DSS Export Volume Flow Curves= 0
DXF OffsetX= 0
DXF OffsetY= 0
DXF ScaleX= 1
DXF ScaleY= 10

--- Forbush Creek.p01 (plan) ---

Plan Title=Floodway Run
Program Version=3.12
Short Identifier=Floodway
Geom File=g01
Flow File=f01
Subcritical Flow
K Sum by GR= 0
Std Step Tol= 0.01
Critical Tol= 0.01
Num of Std Step Trials= 20
Max Error Tol= 0.3
Flow Tol Ratio= 0.001
Split Flow NTrial= 30
Split Flow Tol= 0.02
Split Flow Ratio= 0.02
Log Output Level= 0
Friction Slope Method= 1
Unsteady Friction Slope Method= 2
Unsteady Bridges Friction Slope Method= 1
Parabolic Critical Depth
Global Vel Dist= 0 , 0 , 0
Global Log Level= 0
CheckData=True
Encroach Param=-1 ,10,10, 2
Encroach River=Forbush Creek
Encroach Reach=Reach-1
Encroach Node=76861
       1    4820    5011
Encroach Node=76567
       1    4928    5060
Encroach Node=76359
       1    4935    5060
Encroach Node=76000
       1    4934    5030
Encroach Node=75555
       1    4913    5063
Encroach Node=74641
       1    4860    5015
Encroach Node=73589
       1    4895    5017
Encroach Node=72802
       1    4960    5100
Encroach Node=71624
       1    4868    5045
Encroach Node=70458
       1    4964    5074
Encroach Node=70184
       1    4950    5130
Encroach Node=70058
       1    4965    5130
Encroach Node=69694
       1    4970    5104
Encroach Node=69118
       1    4968    5040
Encroach Node=68414
       1    4966    5022
Encroach Node=67885
       1    4985    5030
Encroach Node=67749
       1    4960    5030
Encroach Node=67664
       1    4975    5030
Encroach Node=67304
       1    4949    5045
Encroach Node=66947
       1    4973    5038
Encroach Node=65759
       1    4899    5017
Encroach Node=65006
       1    4955    5080
Encroach Node=63907
       1    4910    5007
Encroach Node=63328
       1    4970    5027
Encroach Node=62662
       1    4980    5018
Encroach Node=61870
       1    4960    5018
Encroach Node=60937
       1    4974    5015
Encroach Node=60146
       1    4970    5028
Encroach Node=59666
       1    4978    5078
Encroach Node=58433
       1    4790    5016
Encroach Node=57072
       1    4888    5029
Encroach Node=56156
       1    4800    5064
Encroach Node=55830
       1    4880    5100
Encroach Node=55635
       1    4900    5086
Encroach Node=55049
       1    4925    5120
Encroach Node=54088
       1    4940    5150
Encroach Node=52821
       1    4780    5030
Encroach Node=51370
       1    4780    5030
Encroach Node=50066
       1    4874    5110
Encroach Node=49241
       1    4983    5154
Encroach Node=48638
       1    4920    5040
Encroach Node=48243
       1    4810    5025
Encroach Node=47414
       1    4840    5035
Encroach Node=46494
       1    4875    5040
Encroach Node=45609
       1    4902    5072
Encroach Node=45322
       1    4908    5075
Encroach Node=45165
       1    4908    5125
Encroach Node=44759
       1    4844    5022
Encroach Node=44279
       1    4942    5060
Encroach Node=43540
       1    4960    5030
Encroach Node=42902
       1    4950    5124
Encroach Node=42360
       1    4981    5070
Encroach Node=41368
       1    4870    5025
Encroach Node=40679
       1    4892    5020
Encroach Node=40445
       1    4855    5084
Encroach Node=40280
       1    4841    5081
Encroach Node=40006
       1    4840    5040
Encroach Node=39135
       1    4780    5100
Encroach Node=38320
       1    4900    5140
Encroach Node=37748
       1    4942    5067
Encroach Node=37560
       1    4943    5045
Encroach Node=37414
       1    4943    5045
Encroach Node=37119
       1    4964    5120
Encroach Node=36236
       1    4911    5060
Encroach Node=35964
       1    4920    5110
Encroach Node=35849
       1    4942    5120
Encroach Node=35315
       1    4910    5190
Encroach Node=34461
       1    4922    5176
Encroach Node=33705
       1    4760    5100
Encroach Node=32450
       1    4880    5250
Encroach Node=31427
       1    4830    5030
Encroach Node=30468
       1    4740    5044
Encroach Node=29458
       1    4780    5204
Encroach Node=28343
       1    4960    5188
Encroach Node=27395
       1    4822    5024
Encroach Node=26751
       1    4960    5080
Encroach Node=25863
       1    4970    5055
Encroach Node=24860
       1    4947    5022
Encroach Node=24210
       1    4900    5045
Encroach Node=23879
       1    4940    5058
Encroach Node=23755
       1  4898.5  5101.5
Encroach Node=23206
       1    4640    5050
Encroach Node=22043
       1    4930    5125
Encroach Node=21260
       1    4915    5018
Encroach Node=20462
       1    4930    5040
Encroach Node=19679
       1    4948    5140
Encroach Node=18940
       1  4965.6    5358
Encroach Node=17167
       1    4683    5022
Encroach Node=15453
       1    4520    5033
Encroach Node=13527
       1    4770    5050
Encroach Node=12665
       1    4652    5169
Encroach Node=11033
       1    4460    5030
Encroach Node=9393
       1    4730    5058
Encroach Node=7615
       1    4776    5030
Encroach Node=7331
       1    4860    5086
Encroach Node=7063
       1    4870    5130
Encroach Node=6474
       1    4840    5284
Encroach Node=5583
       1    4580    5300
Encroach Node=3684
       1    4640    5230
Encroach Node=3269
       1    4815    5080
Encroach Node=3062
       1    4810    5150
Encroach Node=2543
       1    4940    5490
BEGIN DESCRIPTION:
Floodway Run
END DESCRIPTION:
Computation Interval=1HOUR
Output Interval=1HOUR
Run HTab= 0
Run UNet= 0
Run PostProcess= 0
UNET Theta= 1
UNET Theta Warmup= 1
UNET ZTol= 0.02
UNET ZSATol= 0.05
UNET MxIter= 20
UNET MaxInSteps= 0
UNET DtIC= 0
UNET DtMin= 0
UNET MaxCRTS= 20
UNET WFStab= 2
UNET SFStab= 1
UNET WFX= 1
UNET SFX= 1
UNET DSS MLevel= 4
UNET DZMax Abort= 100
UNET Convert EG Bridges=-1
UNET Use Existing IB Tables=-1
UNET Froude Reduction=False
UNET Froude Limit= 1
UNET Froude Power= 10
Instantaneous Interval=1HOUR
Write IC File= 0
Echo Input=False
Echo Output=False
Write Detailed= 0
Detailed Automatic Start=False, 10

--- Forbush Creek.f01 (steady flow) ---

Flow Title=Floodway
Number of Profiles=2
Profile Names=100-year,100-FW
River Rch & RM= Forbush Creek,Reach-1,76861
    1679    1679
River Rch & RM= Forbush Creek,Reach-1,74641
    1976    1976
River Rch & RM= Forbush Creek,Reach-1,70458
    2056    2056
River Rch & RM= Forbush Creek,Reach-1,67304
    2471    2471
River Rch & RM= Forbush Creek,Reach-1,58433
    2550    2550
River Rch & RM= Forbush Creek,Reach-1,56156
    3061    3061
River Rch & RM= Forbush Creek,Reach-1,52821
    3117    3117
River Rch & RM= Forbush Creek,Reach-1,50066
    3179    3179
River Rch & RM= Forbush Creek,Reach-1,48638
    3183    3183
River Rch & RM= Forbush Creek,Reach-1,48243
    3361    3361
River Rch & RM= Forbush Creek,Reach-1,45322
    3410    3410
River Rch & RM= Forbush Creek,Reach-1,41368
    3510    3510
River Rch & RM= Forbush Creek,Reach-1,39135
    3537    3537
River Rch & RM= Forbush Creek,Reach-1,35315
    3796    3796
River Rch & RM= Forbush Creek,Reach-1,32450
    3817    3817
River Rch & RM= Forbush Creek,Reach-1,27395
    3819    3819
River Rch & RM= Forbush Creek,Reach-1,23206
    4327    4327
River Rch & RM= Forbush Creek,Reach-1,18940
    4517    4517
River Rch & RM= Forbush Creek,Reach-1,15453
    4749    4749
River Rch & RM= Forbush Creek,Reach-1,12665
    4936    4936
River Rch & RM= Forbush Creek,Reach-1,6474
    9002    9002
Boundary for River Rch & Prof#=Forbush Creek,Reach-1,1
Up Type=0
Dn Type=3
Dn Slope=0.001
Boundary for River Rch & Prof#=Forbush Creek,Reach-1,2
Up Type=0
Dn Type=3
Dn Slope=0.001

--- Forbush Creek.g01 (geometry) ---

Geom Title=Existing Conditions

River Reach=Forbush Creek,Reach-1
Reach XY= 30
      1518560.00       896247.88      1521551.27       888814.72
      1522084.75       888324.59      1523376.80       888856.22
      1522950.60       887946.48      1523668.05       887843.26
      1524893.95       885945.92      1524624.64       884021.91
      1522820.57       882853.78      1522292.18       880911.25
      1526331.77       878782.81      1528074.96       880614.73
      1529202.24       879788.98      1530450.77       879748.55
      1532381.45       880945.85      1533775.05       880221.27
      1535351.41       878978.69      1535376.54       877374.79
      1536381.09       877565.70      1536592.88       875158.25
      1538671.22       874274.01      1538712.89       872732.35
      1544083.63       871398.50      1543757.76       870826.38
      1544744.78       868800.37      1549601.40       867393.38
      1550815.25       866021.00      1554224.13       867366.88
      1554682.19       866798.41      1554522.50       860880.25

Type RM Length L Ch R = 1,76861,294,294,294
BEGIN DESCRIPTION:
Forbush Creek - 81.0
END DESCRIPTION:
XS GIS Cut Line= 4
      1519613.84       895346.84      1519299.45       895276.26
      1518920.93       895038.89      1518670.71       895109.46
#Sta/Elev= 30
  4265.8  969.84  4330.5  963.60  4352.1  959.46  4398.4  954.80  4456.8  945.53
  4507.6  935.67  4579.9  921.90  4627.8  919.27  4640.9  917.60  4642.5  915.79
  4642.7  916.73  4654.9  918.48  4676.5  919.10  4821.5  917.15  4974.8  919.20
  4993.3  919.00  4997.2  914.62  4998.7  911.62  5001.3  911.62  5002.8  914.62
  5011.0  920.25  5013.6  926.56  5042.9  928.73  5049.9  927.36  5081.0  930.37
  5103.8  932.22  5138.3  938.35  5219.4  948.82  5253.1  952.12  5294.8  953.67
#Mann=7,-1,0
  4265.8    0.08       0  4507.6    0.14       0  4676.5    0.08       0
  4974.8    0.14       0  4997.2    0.05       0  5002.8    0.14       0
  5081.0    0.08       0
Bank Sta=4997.2,5002.8
XS Rating Curve= 0
Exp/Cntr=0.5,0.3

Type RM Length L Ch R = 1,76567,208,208,208
BEGIN DESCRIPTION:
Union Grove Church Road  FC - us
END DESCRIPTION:
XS GIS Cut Line= 4
      1519649.09       895314.75      1519302.66       895022.85
      1518985.09       894657.16      1518799.04       894172.81
#Sta/Elev= 30
  4307.4  971.05  4413.8  962.63  4531.5  944.59  4557.6  945.01  4591.2  942.05
  4616.0  936.58  4743.5  920.15  4817.8  917.61  4848.6  914.31  4888.6  917.37
  4917.6  915.82  4987.4  917.00  4987.8  911.50  5011.6  911.50  5012.6  914.18
  5076.1  921.06  5148.8  922.41  5170.6  923.19  5231.4  932.37  5279.6  936.42
  5318.3  941.87  5356.8  953.23  5380.0  958.49  5443.5  959.63  5475.7  957.66
  5583.1  964.15  5603.5  963.93  5649.5  977.13  5669.9  977.10  5763.6  985.10
#Mann=8,-1,0
  4307.4    0.08       0  4817.8    0.14       0  4987.4    0.05       0
  5012.6    0.14       0  5148.8    0.08       0  5279.6    0.14       0
  5356.8    0.08       0  5583.1    0.08       0
#XS Ineff=2,0
    0.00 4926.50  940.20 5073.50    0.00  940.20
Permanent Ineff=
       F       F
Bank Sta=4987.4,5012.6
XS Rating Curve= 0
Exp/Cntr=0.5,0.3

Type RM Length L Ch R =2,76465,,,
BEGIN DESCRIPTION:
Union Grove Church Road  FC - TOR
Structure ID: LDS_FC_12
Approximate Survey Structure
END DESCRIPTION:
Bridge Culvert--1,0,-1,-1,0
Deck Dist Width WeirC Skew NumUp NumDn MinLoCord MaxHiCord MaxSubmerge Is_Ogee
62,80,3,,9,9,,,0.95,0,1,1,,,
  4271.4  4352.9  4504.6  4657.3  4793.9  5080.4  5177.3  5319.4  5784.7
  972.91  968.08  952.89  945.30  940.20  940.20  942.52  948.81  988.93
  891.50  891.50  891.50  891.50  891.50  891.50  891.50  891.50  891.50
  4271.4  4352.9  4504.6  4657.3  4793.9  5080.4  5177.3  5319.4  5784.7
  972.91  968.08  952.89  945.30  940.20  940.20  942.52  948.81  988.93
  891.10  891.10  891.10  891.10  891.10  891.10  891.10  891.10  891.10
Culvert=2,9,11,80,0.012,0.4,1,8,1,911.7,4994,911.3,4994,Culvert #1,0,62
Culvert Bottom n=0.012
Culvert Bottom Depth=0
Culvert Depth Blocked=0
Culvert=2,9,11,80,0.012,0.4,1,8,1,911.7,5006,911.3,5006,Culvert #2,0,62
Culvert Bottom n=0.012
Culvert Bottom Depth=0
Culvert Depth Blocked=0
BC Design=,,0,,0,,,,,,

Type RM Length L Ch R = 1,76359,359,359,359
BEGIN DESCRIPTION:
Union Grove Church Road  FC - ds
END DESCRIPTION:
XS GIS Cut Line= 4
      1519716.47       895250.61      1519549.66       894945.86
      1519062.07       894474.32      1518840.74       894143.92
#Sta/Elev= 30
  4277.8  970.44  4360.7  964.48  4444.9  953.52  4559.6  948.21  4620.7  942.72
  4670.7  939.86  4679.0  937.84  4719.9  933.34  4806.9  925.83  4881.3  917.58
  4937.3  916.60  4956.1  917.73  4987.4  915.27  4988.0  911.10  5012.1  911.10
  5012.6  914.55  5033.7  918.28  5051.1  917.67  5082.6  919.64  5102.6  919.28
  5138.0  923.05  5148.6  927.38  5168.8  932.96  5188.6  936.95  5199.6  937.26
  5253.8  939.23  5296.2  942.36  5451.3  958.50  5556.8  971.78  5701.2  985.46
#Mann=5,-1,0
  4277.8    0.08       0  4559.6    0.14       0  4987.4    0.05       0
  5012.6    0.14       0  5199.6    0.08       0
#XS Ineff=2,0
    0.00 4922.50  940.20 5077.50    0.00  940.20
Permanent Ineff=
       F       F
Bank Sta=4987.4,5012.6
XS Rating Curve= 0
Exp/Cntr=0.5,0.3

Type RM Length L Ch R = 1,76000,445,445,445
BEGIN DESCRIPTION:
Forbush Creek - 80.0
END DESCRIPTION:
XS GIS Cut Line= 3
      1519947.39       894477.53      1519665.14       894525.64
      1519219.24       894240.13
#Sta/Elev= 30
  4419.0  958.32  4494.8  957.05  4615.4  951.89  4673.0  950.03  4697.0  947.63
  4722.3  943.40  4754.2  935.62  4798.3  926.38  4833.2  920.55  4870.8  917.53
  4876.8  917.59  4903.4  915.21  4945.3  915.26  4953.2  914.51  4989.4  915.12
  4994.4  913.68  4995.4  911.41  4996.8  908.41  5003.2  908.41  5004.6  911.41
  5036.0  915.33  5062.9  926.67  5099.7  937.42  5116.2  942.96  5137.2  948.94
  5147.5  951.79  5161.9  951.59  5167.9  952.14  5204.5  954.22  5234.8  957.20
#Mann=7,-1,0
  4419.0    0.08       0  4615.4    0.14       0  4995.4    0.05       0
  5004.6    0.14       0  5137.2    0.08       0  5167.9    0.14       0
  5204.5    0.08       0
Bank Sta=4995.4,5004.6
XS Rating Curve= 0
Exp/Cntr=0.3,0.1

Type RM Length L Ch R = 1,75555,914,914,914
BEGIN DESCRIPTION:
Forbush Creek - 79.0
END DESCRIPTION:
XS GIS Cut Line= 2
      1519950.65       893957.86      1519132.66       893919.37
#Sta/Elev= 30
  4541.5  949.57  4567.7  948.81  4621.4  945.09  4711.3  936.33  4747.1  931.76
  4795.6  921.87  4819.2  918.44  4841.7  916.23  4857.0  915.66  4877.1  914.07
  4926.5  911.69  4964.2  913.74  4979.9  913.90  4994.9  908.41  4996.4  905.41
  5003.6  905.41  5005.1  908.41  5011.4  914.58  5016.4  914.43  5058.1  913.21
  5085.2  913.27  5100.3  914.35  5107.8  915.42  5112.9  916.99  5134.7  923.25
  5153.9  929.95  5195.4  940.84  5239.8  951.68  5272.1  959.17  5360.4  973.89
#Mann=11,-1,0
  4541.5    0.08       0  4857.0     0.1       0  4926.5    0.08       0
  4964.2    0.14       0  4994.9    0.05       0  5005.1    0.14       0
  5016.4    0.08       0  5112.9    0.14       0  5195.4    0.08       0
  5239.8    0.14       0  5272.1    0.08       0
Bank Sta=4994.9,5005.1
XS Rating Curve= 0
Exp/Cntr=0.3,0.1

Type RM Length L Ch R = 1,74641,1052,1052,1052
BEGIN DESCRIPTION:
Forbush Creek - 78.0
END DESCRIPTION:
XS GIS Cut Line= 3
      1520239.34       893101.38      1519507.96       893062.89
      1519328.36       892921.77
#Sta/Elev= 30
  4361.8  947.23  4456.6  940.03  4498.2  935.88  4542.4  929.86  4568.1  927.87
  4601.8  923.31  4661.6  913.19  4679.4  914.30  4694.4  912.21  4697.0  910.76
  4697.4  912.27  4701.2  912.52  4744.0  911.44  4770.7  909.95  4854.4  909.07
  4954.8  909.12  4983.5  910.01  4989.0  909.71  4994.9  904.67  4996.4  901.67
  5003.6  901.67  5005.1  904.67  5013.3  911.43  5056.8  918.14  5124.1  937.54
  5146.4  942.54  5171.9  945.45  5228.5  952.44  5256.5  954.73  5322.6  958.40
#Mann=5,-1,0
  4361.8    0.08       0  4601.8    0.14       0  4994.9    0.05       0
  5005.1    0.14       0  5171.9    0.08       0
#XS Ineff=2,0
    0.00 4680.10  926.50               0
Permanent Ineff=
       F       F
Bank Sta=4994.9,5005.1
XS Rating Curve= 0
Exp/Cntr=0.3,0.1

Type RM Length L Ch R = 1,73589,787,787,787
BEGIN DESCRIPTION:
Forbush Creek - 77.0
END DESCRIPTION:
XS GIS Cut Line= 4
      1520560.12       892549.65      1520402.93       892337.93
      1519957.05       892161.50      1519690.81       892139.04
#Sta/Elev= 30
  4308.1  946.71  4393.7  938.52  4500.0  929.32  4541.0  927.87  4582.7  922.79
  4718.9  913.38  4771.9  908.62  4803.8  906.98  4848.5  905.67  4954.0  906.10
  4964.3  904.93  4974.2  904.73  4983.8  902.04  4993.3  900.45  4994.8  897.45
  5005.2  897.45  5006.7  900.45  5019.1  906.73  5025.7  906.24  5057.5  906.75
  5067.0  909.31  5077.9  914.75  5090.5  918.53  5108.2  925.03  5123.1  928.38
  5153.7  933.75  5225.8  943.58  5248.0  944.34  5268.7  947.73  5318.5  950.54
#Mann=4,-1,0
  4308.1    0.08       0  4954.0    0.14       0  4993.3    0.05       0
  5006.7    0.14       0
Bank Sta=4993.3,5006.7
XS Rating Curve= 0
Exp/Cntr=0.3,0.1

Type RM Length L Ch R = 1,72802,1178,1178,1178
BEGIN DESCRIPTION:
Forbush Creek - 76.0
END DESCRIPTION:
XS GIS Cut Line= 2
      1520771.83       891680.33      1520005.17       891346.72
#Sta/Elev= 30
  4533.9  932.52  4580.1  928.15  4592.4  926.07  4645.1  920.91  4844.6  909.50
  4898.1  905.46  4921.5  902.85  4964.8  902.11  4966.5  901.60  4979.1  898.55
  4993.3  897.50  4994.8  894.50  5005.2  894.50  5006.7  897.50  5010.8  901.71
  5013.2  905.58  5020.6  906.17  5026.2  904.76  5032.3  903.77  5086.9  903.89
  5162.8  902.91  5189.1  902.84  5201.7  903.59  5223.2  912.79  5234.9  920.60
  5279.9  933.91  5291.2  937.93  5306.2  941.44  5326.8  944.24  5370.0  951.03
#Mann=7,-1,0
  4533.9    0.08       0  4966.5    0.14       0  4993.3    0.05       0
  5006.7    0.14       0  5026.2    0.08       0  5162.8    0.14       0
  5326.8    0.08       0
Bank Sta=4993.3,5006.7
XS Rating Curve= 0
Exp/Cntr=0.3,0.1

Type RM Length L Ch R = 1,71624,1166,1166,1166
BEGIN DESCRIPTION:
Forbush Creek - 75.0
END DESCRIPTION:
XS GIS Cut Line= 3
      1521230.56       890766.15      1521137.52       890547.98
      1520511.96       890336.25
#Sta/Elev= 30
  4395.5  936.32  4459.7  931.62  4480.7  930.69  4558.9  922.38  4625.0  910.52
  4659.1  905.99  4681.8  904.15  4733.8  901.85  4866.1  900.18  4939.9  900.35
  4957.6  897.56  4986.4  896.97  4993.3  893.72  4994.8  890.72  5005.2  890.72
  5006.7  893.72  5017.1  897.46  5025.6  897.25  5040.7  894.60  5054.8  902.08
  5082.5  903.91  5085.7  904.28  5099.5  910.32  5109.2  912.09  5122.2  916.36
  5143.8  920.81  5151.5  923.14  5200.4  931.70  5223.0  933.30  5293.1  940.62
#Mann=9,-1,0
  4395.5    0.08       0  4459.7    0.14       0  4659.1    0.08       0
  4957.6    0.14       0  4993.3    0.05       0  5006.7    0.14       0
  5025.6    0.08       0  5082.5    0.14       0  5223.0    0.08       0
Bank Sta=4993.3,5006.7
XS Rating Curve= 0
Exp/Cntr=0.3,0.1

Type RM Length L Ch R = 1,70458,274,274,274
BEGIN DESCRIPTION:
Forbush Creek - 74.0
END DESCRIPTION:
XS GIS Cut Line= 4
      1521705.29       889457.33      1521467.92       889479.78
      1521038.07       889325.81      1520771.81       889322.60
#Sta/Elev= 30
  4489.8  933.44  4603.6  920.50  4623.8  919.82  4638.5  916.97  4668.9  913.37
  4681.5  913.75  4691.0  911.41  4739.1  908.21  4745.1  904.44  4754.3  903.01
  4854.8  899.10  4882.1  900.61  4917.9  897.66  4941.2  897.88  4954.0  899.20
  4979.1  897.35  4993.0  892.53  4994.5  889.53  5005.5  889.53  5007.0  892.53
  5017.1  898.53  5026.4  898.37  5066.7  897.12  5110.7  897.75  5159.2  900.35
  5168.3  900.63  5189.1  906.25  5212.6  909.65  5261.7  914.06  5451.1  932.50
#Mann=9,-1,0
  4489.8    0.14       0  4754.3    0.08       0  4882.1    0.14       0
  4993.0    0.05       0  5007.0    0.14       0  5026.4    0.08       0
  5159.2    0.14       0  5212.6    0.08       0  5261.7    0.14       0
#XS Ineff=2,0
    0.00 4884.50  907.75               0
Permanent Ineff=
       F       F
Bank Sta=4993,5007
XS Rating Curve= 0
Exp/Cntr=0.5,0.3

Type RM Length L Ch R = 1,70184,126,126,126
BEGIN DESCRIPTION:
Private Drive 2  FC - us
END DESCRIPTION:
XS GIS Cut Line= 4
      1521641.11       889354.66      1521243.37       889091.64
      1521111.85       889059.56      1520941.82       889043.52
#Sta/Elev= 30
  4714.7  928.28  4780.9  920.20  4819.3  912.86  4825.9  912.49  4864.9  905.31
  4871.3  905.39  4880.3  902.82  4887.0  900.84  4894.0  900.19  4940.8  898.37
  4971.2  897.99  4975.2  896.96  4982.0  896.60  4988.8  889.00  5011.3  889.00
  5018.0  896.60  5024.7  897.65  5046.6  896.98  5129.9  897.43  5169.4  897.00
  5279.5  898.46  5302.3  899.52  5323.1  902.94  5345.5  903.55  5361.6  907.80
  5401.7  914.03  5419.0  916.49  5453.8  920.04  5471.0  922.86  5497.7  926.04
#Mann=7,-1,0
  4714.7    0.14       0  4880.3    0.08       0  4940.8    0.14       0
  4982.0    0.05       0  5018.0    0.14       0  5279.5    0.14       0
  5453.8    0.08       0
#XS Ineff=2,0
    0.00 4919.80  898.05 5080.30    0.00  896.63
Permanent Ineff=
       F       F
Bank Sta=4982,5018
XS Rating Curve= 0
Exp/Cntr=0.5,0.3

Type RM Length L Ch R =3,70112,,,
BEGIN DESCRIPTION:
Private Drive 2  FC - TOR
Structure ID: LDS_FC_10
Approximate Survey Structure
END DESCRIPTION:
Bridge Culvert--1,0,-1,-1,0
Deck Dist Width WeirC Skew NumUp NumDn MinLoCord MaxHiCord MaxSubmerge Is_Ogee
65.5,13,3,,13,13,,,0.95,0,1,1,,,
  4722.8  4856.0  4903.0  4924.4  4985.3  4985.3  5014.8  5014.8  5035.7  5144.4
  5263.4  5444.0  5575.8
  929.08  911.33  905.62  900.41  898.50  898.50  898.50  898.50  898.41  896.82
  897.92  912.91  927.07
  869.00  869.00  869.00  869.00  869.00  896.00  896.00  869.00  869.00  869.00
  869.00  869.00  869.00
  4722.8  4856.0  4903.0  4924.4  4985.3  4985.3  5014.8  5014.8  5035.7  5144.4
  5263.4  5444.0  5575.8
  929.08  911.33  905.62  900.41  898.50  898.50  898.50  898.50  898.41  896.82
  897.92  912.91  927.07
  869.00  869.00  869.00  869.00  869.00  896.00  896.00  869.00  869.00  869.00
  869.00  869.00  869.00
BR Coef=1,1,0,1.25,0,,,0.8,0,2,0,
WSPro=,,,, 1 ,,,, 0 ,,,, 0 ,,,,-1 ,-1 ,-1 , 0 , 0 , 0 , 0 , 0
BC Design=,,0,,0,,,,,,

Type RM Length L Ch R = 1,70058,364,364,364
BEGIN DESCRIPTION:
Private Drive 2  FC - ds
END DESCRIPTION:
XS GIS Cut Line= 4
      1521705.33       889236.01      1521281.87       888979.37
      1521134.31       888953.71      1520935.43       888992.20
#Sta/Elev= 30
  4740.9  931.31  4793.0  925.00  4837.0  918.40  4858.0  916.22  4881.0  911.94
  4901.9  909.12  4912.7  905.79  4929.2  900.71  4944.4  900.19  4953.1  899.22
  4965.4  897.82  4984.5  897.30  4985.7  896.35  4991.3  888.75  5011.3  888.75
  5023.1  894.05  5037.7  895.86  5120.7  896.56  5148.2  895.82  5225.2  896.60
  5287.0  896.34  5336.2  898.75  5348.3  900.54  5376.4  902.67  5420.9  908.38
  5489.0  914.12  5526.5  919.25  5547.1  920.70  5555.6  920.60  5588.4  924.02
#Mann=7,-1,0
  4740.9    0.14       0  4912.7    0.08       0  4953.1    0.14       0
  4985.7    0.05       0  5023.1    0.14       0  5037.7    0.08       0
  5348.3    0.14       0
#XS Ineff=2,0
    0.00 4937.80  897.78 5062.30    0.00  896.79
Permanent Ineff=
       F       F
Bank Sta=4985.7,5023.1
XS Rating Curve= 0
Exp/Cntr=0.5,0.3

Type RM Length L Ch R = 1,69694,576,576,576
BEGIN DESCRIPTION:
Forbush Creek - 73.0
END DESCRIPTION:
XS GIS Cut Line= 3
      1521894.58       888950.51      1521352.44       888626.51
      1521076.58       888562.36
#Sta/Elev= 30
  4649.3  927.58  4667.6  927.08  4695.8  922.09  4731.7  920.06  4787.7  915.73
  4803.9  910.06  4826.5  910.58  4888.5  902.69  4909.6  900.82  4955.2  898.43
  4965.6  897.59  4970.3  895.65  4993.0  889.61  4994.5  886.61  5005.5  886.61
  5007.0  889.61  5026.2  890.68  5050.0  893.91  5057.0  893.88  5123.2  895.12
  5204.8  895.04  5257.4  897.08  5283.9  898.24  5310.3  903.31  5319.5  904.20
  5334.2  907.18  5362.2  911.48  5424.4  919.19  5516.6  930.55  5564.1  938.23
#Mann=10,-1,0
  4649.3    0.14       0  4787.7    0.08       0  4955.2    0.14       0
  4993.0    0.05       0  5007.0    0.14       0  5057.0    0.08       0
  5257.4    0.14       0  5283.9    0.08       0  5319.5    0.14       0
  5424.4    0.08       0
Bank Sta=4993,5007
XS Rating Curve= 0
Exp/Cntr=0.3,0.1

Type RM Length L Ch R = 1,69118,704,704,704
BEGIN DESCRIPTION:
Forbush Creek - 72.0
END DESCRIPTION:
XS GIS Cut Line= 3
      1522048.54       888684.29      1521958.71       888315.36
      1522067.79       888093.99
#Sta/Elev= 30
  4688.8  942.70  4805.6  929.83  4825.4  926.59  4841.0  924.89  4855.3  920.13
  4868.1  917.72  4922.7  900.33  4941.5  896.29  4942.1  893.88  4955.0  891.39
  4961.5  894.43  4987.6  890.05  4993.0  886.39  4994.5  883.39  5005.5  883.39
  5007.0  886.39  5007.6  887.70  5021.3  890.43  5032.8  890.74  5055.8  895.91
  5059.7  896.36  5068.5  899.79  5124.3  916.81  5160.1  925.55  5175.9  927.45
  5192.1  928.58  5228.2  933.02  5240.2  935.87  5249.5  937.04  5315.3  945.68
#Mann=4,-1,0
  4688.8    0.14       0  4993.0    0.05       0  5007.0    0.14       0
  5249.5    0.08       0
Bank Sta=4993,5007
XS Rating Curve= 0
Exp/Cntr=0.3,0.1

Type RM Length L Ch R = 1,68414,529,529,529
BEGIN DESCRIPTION:
Forbush Creek - 71.0
END DESCRIPTION:
XS GIS Cut Line= 2
      1522577.81       888729.19      1522603.48       888244.77
#Sta/Elev= 30
  4761.4  930.03  4767.3  927.82  4778.3  927.76  4792.2  925.08  4822.8  920.23
  4838.3  917.96  4847.4  916.20  4869.2  913.15  4891.2  911.74  4896.2  910.92
  4914.5  903.31  4948.8  891.35  4962.7  887.63  4993.0  883.47  4994.5  880.47
  5005.5  880.47  5007.0  883.47  5038.8  890.64  5054.4  892.74  5069.5  893.61
  5094.9  899.12  5108.6  904.81  5118.8  910.56  5127.9  914.45  5138.4  916.97
  5164.6  925.13  5198.0  934.26  5217.0  938.84  5233.4  942.07  5246.5  943.95
#Mann=5,-1,0
  4761.4    0.08       0  4822.8    0.14       0  4993.0    0.05       0
  5007.0    0.14       0  5164.6    0.08       0
Bank Sta=4993,5007
XS Rating Curve= 0
Exp/Cntr=0.3,0.1

Type RM Length L Ch R = 1,67885,136,136,136
BEGIN DESCRIPTION:
Forbush Creek - 70.0
END DESCRIPTION:
XS GIS Cut Line= 3
      1522821.63       888906.72      1523068.62       888663.53
      1523093.31       888578.05
#Sta/Elev= 30
  4723.4  929.95  4761.3  922.27  4797.4  913.36  4810.7  912.71  4837.4  912.33
  4865.1  907.54  4893.2  901.61  4905.3  899.85  4909.3  898.88  4924.0  897.02
  4929.3  896.22  4942.8  893.24  4947.0  892.92  4973.0  889.03  4985.2  887.95
  4990.5  886.91  4993.0  882.25  4994.5  879.25  5005.5  879.25  5007.0  882.25
  5015.4  883.19  5025.0  885.14  5029.2  885.29  5053.6  889.84  5081.4  893.99
  5096.8  898.53  5106.5  900.88  5125.7  904.29  5137.8  906.87  5159.0  908.90
#Mann=7,-1,0
  4723.4    0.08       0  4865.1    0.14       0  4924.0    0.08       0
  4942.8    0.14       0  4993.0    0.05       0  5007.0    0.14       0
  5106.5    0.08       0
Bank Sta=4993,5007
XS Rating Curve= 0
Exp/Cntr=0.5,0.3

Type RM Length L Ch R = 1,67749,85,85,85
BEGIN DESCRIPTION:
Griffin Road  FC - us
END DESCRIPTION:
XS GIS Cut Line= 3
      1523113.38       889098.41      1523121.72       888698.01
      1523100.02       888586.18
#Sta/Elev= 30
  4702.5  931.05  4705.8  930.46  4729.5  924.14  4750.5  919.91  4766.2  916.10
  4790.4  908.65  4822.9  904.62  4842.9  902.06  4857.4  898.92  4889.5  893.01
  4905.8  891.72  4918.7  891.13  4952.3  887.24  4976.5  886.65  4985.0  885.70
  4988.0  879.00  5012.0  879.00  5015.0  885.70  5033.9  886.81  5049.9  886.99
  5070.8  887.97  5096.4  892.90  5107.6  894.43  5112.1  895.82  5123.2  896.90
  5128.7  897.91  5153.1  900.16  5162.4  902.01  5202.3  906.45  5216.9  907.51
#Mann=5,-1,0
  4702.5    0.14       0  4822.9    0.14       0  4985.0    0.05       0
  5015.0    0.14       0  5162.4    0.08       0
#XS Ineff=2,0
    0.00 4948.50  889.26 5051.50    0.00  889.35
Permanent Ineff=
       F       F
Bank Sta=4985,5015
XS Rating Curve= 0
Exp/Cntr=0.5,0.3

Type RM Length L Ch R =3,67702,,,
BEGIN DESCRIPTION:
Griffin Road  FC - TOR
Structure ID: LDS_FC_09
Approximate Survey Structure
END DESCRIPTION:
Bridge Culvert--1,0,-1,-1,0
Deck Dist Width WeirC Skew NumUp NumDn MinLoCord MaxHiCord MaxSubmerge Is_Ogee
36.5,21,3,,16,16,,,0.95,0,1,1,,,
  4689.6  4775.6  4815.6  4866.7  4881.0  4909.3  4925.2  4980.4  4985.0  4985.0
  5015.0  5015.0  5015.5  5047.5  5132.4  5264.1
  937.44  921.76  909.10  904.16  900.68  891.54  890.35  888.00  888.00  888.00
  888.00  888.00  888.00  888.99  896.70  909.52
  859.00  859.00  859.00  859.00  859.00  859.00  859.00  859.00  859.00  886.00
  886.00  859.00  859.00  859.00  859.00  859.00
  4689.6  4775.6  4815.6  4866.7  4881.0  4909.3  4925.2  4980.4  4985.0  4985.0
  5015.0  5015.0  5015.5  5047.5  5132.4  5264.1
  937.44  921.76  909.10  904.16  900.68  891.54  890.35  888.00  888.00  888.00
  888.00  888.00  888.00  888.99  896.70  909.52
  859.00  859.00  859.00  859.00  859.00  859.00  859.00  859.00  859.00  886.00
  886.00  859.00  859.00  859.00  859.00  859.00
Abutment Skew #Up #Dn=,2,2
  4985.0  4987.0
  886.00  881.23
  4985.0  4987.0
  886.00  880.98
Abutment Skew #Up #Dn=,2,2
  5013.0  5015.0
  881.23  886.00
  5013.0  5015.0
  880.98  886.00
BR Coef=1,1,0,1.25,0,,,0.8,0,2,0,
WSPro=,,,, 1 ,,,, 0 ,,,, 0 ,,,,-1 ,-1 ,-1 , 0 , 0 , 0 , 0 , 0
BC Design=,,0,,0,,,,,,

Type RM Length L Ch R = 1,67664,360,360,360
BEGIN DESCRIPTION:
Griffin Road  FC - ds
END DESCRIPTION:
XS GIS Cut Line= 3
      1523185.12       889103.44      1523200.14       888739.72
      1523116.71       888584.56
#Sta/Elev= 30
  4731.1  929.84  4750.9  925.30  4779.2  921.93  4803.2  913.86  4818.1  909.92
  4856.2  904.70  4872.4  901.44  4898.6  892.08  4912.8  889.66  4959.8  889.28
  4985.0  885.45  4988.0  878.75  5012.0  878.75  5015.0  885.45  5031.7  886.64
  5042.1  887.70  5058.1  887.51  5095.5  898.17  5101.6  897.67  5119.9  898.98
  5137.4  901.95  5148.7  902.67  5165.9  900.75  5169.8  901.59  5181.5  903.05
  5185.1  904.53  5203.5  904.42  5212.5  905.81  5228.5  904.02  5271.3  907.29
#Mann=8,-1,0
  4731.1    0.14       0  4872.4    0.08       0  4898.6    0.14       0
  4985.0    0.05       0  5015.0    0.14       0  5031.7    0.08       0
  5169.8    0.11       0  5228.5    0.08       0
#XS Ineff=2,0
    0.00 4957.50  888.84 5042.50    0.00  888.75
Permanent Ineff=
       F       F
Bank Sta=4985,5015
XS Rating Curve= 0
Exp/Cntr=0.5,0.3

Type RM Length L Ch R = 1,67304,357,357,357
BEGIN DESCRIPTION:
Forbush Creek - 69.0
END DESCRIPTION:
XS GIS Cut Line= 3
      1523652.87       888632.20      1523320.20       888749.08
      1523140.37       888614.21
#Sta/Elev= 30
  4730.1  942.91  4751.7  939.16  4768.7  936.60  4783.2  932.07  4791.2  930.45
  4859.9  912.38  4905.5  895.39  4918.4  889.72  4933.9  884.92  4947.1  882.26
  4953.9  882.30  4992.7  879.79  4994.1  876.79  5005.9  876.79  5007.3  879.79
  5014.5  883.47  5022.1  884.27  5075.1  887.11  5098.1  889.96  5155.2  898.56
  5177.0  900.32  5204.3  901.92  5223.9  904.43  5234.1  904.80  5242.8  904.45
  5294.5  907.76  5301.8  906.21  5305.1  906.78  5307.3  906.54  5307.5  906.52
#Mann=7,-1,0
  4730.1    0.08       0  4751.7    0.14       0  4992.7    0.05       0
  5007.3    0.14       0  5022.1    0.08       0  5177.0    0.11       0
  5307.3    0.08       0
Bank Sta=4992.7,5007.3
XS Rating Curve= 0
Exp/Cntr=0.3,0.1

Type RM Length L Ch R = 1,66947,1188,1188,1188
BEGIN DESCRIPTION:
Forbush Creek - 68.0
END DESCRIPTION:
XS GIS Cut Line= 2
      1523468.52       888268.07      1523059.45       888524.30
#Sta/Elev= 30
  4731.4  920.22  4747.1  919.70  4789.3  916.75  4841.8  911.52  4858.6  910.36
  4875.8  906.45  4889.9  903.94  4920.5  896.90  4935.5  892.35  4961.8  883.34
  4976.8  880.04  4992.7  878.41  4994.1  875.41  5005.9  875.41  5007.3  878.41
  5016.8  879.18  5023.4  881.13  5030.5  883.20  5042.3  883.75  5053.0  885.01
  5061.6  887.78  5068.0  890.94  5083.5  895.76  5099.5  901.27  5108.6  902.62
  5122.1  906.09  5154.8  912.79  5169.3  915.23  5212.2  914.57  5214.1  914.53
#Mann=8,-1,0
  4731.4    0.08       0  4841.8    0.14       0  4992.7    0.05       0
  5007.3    0.14       0  5023.4    0.08       0  5042.3    0.11       0
  5154.8    0.08       0  5212.2    0.14       0
Bank Sta=4992.7,5007.3
XS Rating Curve= 0
Exp/Cntr=0.3,0.1

Type RM Length L Ch R = 1,65759,753,753,753
BEGIN DESCRIPTION:
Forbush Creek - 67.0
END DESCRIPTION:
XS GIS Cut Line= 3
      1523509.02       888303.99      1523531.50       887796.00
      1523360.68       887616.19
#Sta/Elev= 30
  4573.4  927.79  4612.8  924.36  4643.3  920.14  4659.3  918.15  4680.3  913.75
  4727.1  906.65  4746.4  901.93  4793.4  892.83  4829.3  884.24  4897.4  879.01
  4930.6  880.91  4952.2  878.58  4974.5  877.58  4981.5  874.33  4992.7  873.50
  4994.1  870.50  5005.9  870.50  5007.3  873.50  5013.5  879.54  5027.5  881.61
  5050.0  880.60  5067.3  884.73  5071.2  887.26  5087.9  891.31  5113.1  901.55
  5150.4  912.13  5234.2  931.12  5270.8  936.28  5293.8  938.46  5329.9  939.29
#Mann=4,-1,0
  4573.4    0.08       0  4643.3    0.14       0  4992.7    0.05       0
  5007.3    0.14       0
Bank Sta=4992.7,5007.3
XS Rating Curve= 0
Exp/Cntr=0.3,0.1

Type RM Length L Ch R = 1,65006,1099,1099,1099
BEGIN DESCRIPTION:
Forbush Creek - 66.0
END DESCRIPTION:
XS GIS Cut Line= 2
      1524331.72       887400.38      1523441.62       887270.01
#Sta/Elev= 30
  4639.6  934.23  4688.9  930.36  4729.8  924.74  4780.4  920.01  4824.8  913.51
  4868.4  905.28  4905.0  894.73  4935.6  882.65  4942.5  880.81  4958.2  876.63
  4973.9  874.45  4994.3  871.19  4995.4  868.19  5004.6  868.19  5005.7  871.19
  5011.6  878.49  5017.6  879.81  5045.5  879.41  5090.2  880.42  5136.3  879.08
  5150.5  880.53  5177.9  880.83  5196.9  882.35  5216.8  884.49  5347.0  902.95
  5355.8  902.92  5379.0  905.43  5474.2  917.12  5499.9  918.98  5539.2  923.78
#Mann=5,-1,0
  4639.6    0.14       0  4942.5    0.08       0  4973.9    0.14       0
  4994.3    0.05       0  5005.7    0.14       0
Bank Sta=4994.3,5005.7
XS Rating Curve= 0
Exp/Cntr=0.3,0.1

Type RM Length L Ch R = 1,63907,579,579,579
BEGIN DESCRIPTION:
Forbush Creek - 65.0
END DESCRIPTION:
XS GIS Cut Line= 3
      1524848.77       886505.74      1524385.67       886460.78
      1524133.91       886276.46
#Sta/Elev= 30
  4644.7  921.46  4667.8  919.23  4754.6  908.37  4786.8  902.53  4803.0  898.86
  4857.3  880.68  4870.7  877.13  4895.4  873.67  4923.5  873.77  4970.2  875.63
  4995.1  867.54  4996.0  864.54  5004.0  864.54  5004.9  867.54  5008.4  877.06
  5075.5  889.78  5110.0  892.45  5127.7  895.56  5148.3  897.31  5184.1  898.13
  5193.5  899.30  5199.7  898.50  5229.4  900.48  5249.3  904.00  5272.1  905.63
  5329.2  912.31  5361.9  917.36  5370.3  920.31  5381.5  919.21  5422.0  924.79
#Mann=5,-1,0
  4644.7    0.08       0  4786.8    0.14       0  4995.1    0.05       0
  5004.9    0.14       0  5272.1    0.08       0
Bank Sta=4995.1,5004.9
XS Rating Curve= 0
Exp/Cntr=0.3,0.1

Type RM Length L Ch R = 1,63328,666,666,666
BEGIN DESCRIPTION:
Forbush Creek - 64.0
END DESCRIPTION:
XS GIS Cut Line= 3
      1524812.76       886316.91      1524700.37       885961.76
      1524363.20       885921.30
#Sta/Elev= 30
  4696.6  914.69  4743.5  908.41  4771.4  903.53  4861.9  887.19  4889.8  880.86
  4916.3  873.80  4931.7  870.51  4950.4  867.42  4964.5  866.34  4970.9  865.45
  4989.6  861.28  4993.5  861.22  4994.7  858.22  5005.3  858.22  5006.5  861.22
  5016.1  865.10  5018.0  865.50  5021.1  866.76  5066.8  878.57  5091.1  881.03
  5118.0  884.62  5149.0  890.65  5181.5  894.48  5198.3  897.12  5208.8  897.97
  5222.4  897.70  5234.0  898.36  5251.2  898.17  5266.2  898.79  5408.7  908.53
#Mann=7,-1,0
  4696.6    0.08       0  4771.4    0.14       0  4889.8    0.08       0
  4950.4    0.14       0  4993.5    0.05       0  5006.5    0.14       0
  5266.2    0.08       0
Bank Sta=4993.5,5006.5
XS Rating Curve= 0
Exp/Cntr=0.3,0.1

Type RM Length L Ch R = 1,62662,792,792,792
BEGIN DESCRIPTION:
Forbush Creek - 63.0
END DESCRIPTION:
XS GIS Cut Line= 3
      1524880.16       885633.57      1524709.36       885584.13
      1524273.28       885813.41
#Sta/Elev= 30
  4617.0  912.19  4667.9  909.51  4684.9  906.77  4699.9  903.66  4755.1  895.60
  4765.0  893.53  4779.8  891.68  4794.8  889.12  4822.2  886.33  4838.9  885.31
  4862.0  878.99  4879.9  875.44  4902.1  869.28  4910.9  868.03  4917.8  865.72
  4929.9  863.68  4975.0  860.63  4982.8  858.22  4990.3  857.52  4992.7  855.39
  4994.1  852.39  5005.9  852.39  5007.3  855.39  5054.7  874.45  5073.1  880.30
  5110.1  884.39  5212.8  895.17  5230.1  898.36  5266.0  899.15  5287.5  901.04
#Mann=4,-1,0
  4617.0    0.14       0  4992.7    0.05       0  5007.3    0.14       0
  5110.1    0.08       0
Bank Sta=4992.7,5007.3
XS Rating Curve= 0
Exp/Cntr=0.3,0.1

Type RM Length L Ch R = 1,61870,933,933,933
BEGIN DESCRIPTION:
Forbush Creek - 62.0
END DESCRIPTION:
XS GIS Cut Line= 3
      1525073.52       884905.28      1524601.47       884968.22
      1524462.10       884990.70
#Sta/Elev= 30
  4569.2  918.78  4620.0  915.17  4683.5  906.77  4696.6  906.41  4699.2  905.63
  4709.7  901.13  4718.5  901.15  4734.8  898.32  4744.7  898.54  4753.2  895.98
  4781.8  891.63  4790.8  890.51  4798.7  888.05  4828.0  881.37  4854.0  874.01
  4885.4  867.91  4904.6  860.86  4923.0  858.92  4960.5  853.05  4984.8  852.73
  4991.9  849.53  4993.4  846.53  5006.6  846.53  5008.1  849.53  5038.8  858.57
  5085.5  867.73  5108.8  877.54  5168.3  895.00  5175.2  896.38  5186.6  896.32
#Mann=6,-1,0
  4569.2    0.08       0  4699.2    0.14       0  4781.8    0.08       0
  4798.7    0.14       0  4991.9    0.05       0  5008.1    0.14       0
Bank Sta=4991.9,5008.1
XS Rating Curve= 0
Exp/Cntr=0.3,0.1

Type RM Length L Ch R = 1,60937,791,791,791
BEGIN DESCRIPTION:
Forbush Creek - 61.0
END DESCRIPTION:
XS GIS Cut Line= 2
      1525073.53       884141.01      1524417.15       884365.80
#Sta/Elev= 30
  4625.4  927.46  4679.7  923.36  4705.1  922.17  4740.5  917.66  4773.6  912.57
  4814.5  904.34  4881.1  889.19  4899.2  883.21  4933.2  868.38  4949.4  856.99
  4961.5  850.55  4986.8  846.29  4991.9  842.73  4993.4  839.73  5006.6  839.73
  5008.1  842.73  5009.7  848.34  5009.8  849.73  5022.9  850.47  5060.5  855.12
  5079.5  860.01  5094.9  862.16  5100.7  863.39  5148.8  875.36  5160.2  877.33
  5173.6  880.53  5187.5  883.04  5200.6  886.11  5225.3  889.45  5319.2  904.32
#Mann=3,-1,0
  4625.4    0.14       0  4991.9    0.05       0  5008.1    0.14       0
Bank Sta=4991.9,5008.1
XS Rating Curve= 0
Exp/Cntr=0.3,0.1

Type RM Length L Ch R = 1,60146,480,480,480
BEGIN DESCRIPTION:
Forbush Creek - 60.0
END DESCRIPTION:
XS GIS Cut Line= 3
      1524241.83       883655.45      1524070.98       883979.17
      1524160.89       884235.41
#Sta/Elev= 30
  4746.6  874.96  4837.5  863.39  4850.8  862.25  4860.7  860.06  4880.6  857.01
  4900.4  855.02  4912.5  852.76  4954.3  841.56  4978.6  837.00  4991.9  836.05
  4993.4  833.05  5006.6  833.05  5008.1  836.05  5019.9  841.62  5035.9  842.31
  5054.4  846.26  5064.4  847.42  5089.1  853.69  5114.4  861.70  5140.8  868.69
  5158.4  872.04  5170.1  875.47  5207.5  883.27  5232.0  886.06  5257.5  890.84
  5315.3  898.95  5328.2  903.56  5340.7  903.42  5373.9  907.53  5384.2  907.93
#Mann=4,-1,0
  4746.6    0.08       0  4850.8    0.14       0  4991.9    0.05       0
  5008.1    0.14       0
Bank Sta=4991.9,5008.1
XS Rating Curve= 0
Exp/Cntr=0.3,0.1

Type RM Length L Ch R = 1,59666,1233,1233,1233
BEGIN DESCRIPTION:
Forbush Creek - 59.0
END DESCRIPTION:
XS GIS Cut Line= 4
      1524403.67       883273.35      1523886.65       883394.73
      1523661.87       883704.93      1523598.92       884100.60
#Sta/Elev= 30
  4241.2  876.82  4290.4  872.63  4314.0  871.93  4352.9  868.97  4412.1  867.12
  4464.3  863.33  4612.3  858.15  4722.1  856.01  4821.2  849.87  4923.2  844.94
  4937.4  845.29  4952.7  843.42  4970.9  836.63  4991.9  833.28  4993.4  830.28
  5006.6  830.28  5008.1  833.28  5013.8  833.44  5031.1  837.96  5064.5  837.49
  5103.1  839.42  5231.7  841.92  5283.2  846.52  5299.2  849.01  5334.3  856.63
  5361.5  864.07  5387.8  868.93  5405.6  871.65  5468.2  877.64  5556.0  884.09
#Mann=7,-1,0
  4241.2    0.08       0  4923.2    0.14       0  4991.9    0.05       0
  5008.1    0.14       0  5103.1    0.08       0  5299.2    0.14       0
  5468.2    0.08       0
#XS Ineff=2,0
       0                 5105.00    0.00  855.54
Permanent Ineff=
       F       F
Bank Sta=4991.9,5008.1
XS Rating Curve= 0
Exp/Cntr=0.3,0.1

Type RM Length L Ch R = 1,58433,1361,1361,1361
BEGIN DESCRIPTION:
Forbush Creek - 58.0
END DESCRIPTION:
XS GIS Cut Line= 4
      1523468.58       882563.03      1523279.74       882581.02
      1522722.27       882895.71      1522466.00       883381.28
#Sta/Elev= 30
  4276.4  884.10  4345.6  869.92  4465.0  839.68  4488.0  838.22  4652.1  832.52
  4776.6  832.34  4829.2  833.05  4891.4  832.58  4947.7  833.41  4967.7  832.45
  4992.1  827.94  4993.4  826.58  4994.6  823.58  5005.4  823.58  5006.6  826.58
  5022.3  835.57  5096.6  851.91  5114.0  853.45  5152.5  850.72  5205.1  851.61
  5229.3  851.76  5242.6  853.56  5309.7  856.24  5343.9  859.02  5392.7  865.16
  5411.9  866.62  5468.7  867.29  5497.3  874.10  5513.5  875.99  5655.3  880.07
#Mann=9,-1,0
  4276.4    0.14       0  4488.0    0.08       0  4776.6    0.14       0
  4829.2    0.08       0  4891.4    0.14       0  4993.4    0.05       0
  5006.6    0.14       0  5205.1     0.1       0  5392.7    0.14       0
Bank Sta=4993.4,5006.6
XS Rating Curve= 0
Exp/Cntr=0.3,0.1

Type RM Length L Ch R = 1,57072,916,916,916
BEGIN DESCRIPTION:
Forbush Creek - 57.0
END DESCRIPTION:
XS GIS Cut Line= 3
      1522681.81       881632.43      1522142.33       881726.84
      1521931.03       882099.99
#Sta/Elev= 30
  4556.6  902.29  4634.5  894.36  4648.2  892.61  4659.6  890.13  4677.5  889.43
  4693.8  884.72  4733.9  875.40  4766.0  865.58  4808.5  850.90  4843.5  837.20
  4869.6  829.45  4878.2  827.25  4901.3  826.51  4924.5  828.46  4935.2  825.71
  4958.4  832.83  4979.8  827.02  4984.8  826.63  4992.5  821.88  4993.9  818.88
  5006.1  818.88  5007.5  821.88  5027.3  826.74  5052.5  827.34  5071.4  829.59
  5118.1  838.43  5220.6  843.22  5244.2  845.24  5358.9  851.89  5533.1  857.59
#Mann=6,-1,0
  4556.6    0.14       0  4869.6    0.08       0  4901.3    0.14       0
  4992.5    0.05       0  5007.5    0.14       0  5244.2    0.08       0
Bank Sta=4992.5,5007.5
XS Rating Curve= 0
Exp/Cntr=0.3,0.1

Type RM Length L Ch R = 1,56156,326,326,326
BEGIN DESCRIPTION:
Forbush Creek - 56.0
END DESCRIPTION:
XS GIS Cut Line= 3
      1522704.31       881452.63      1522214.26       880751.27
      1521953.48       880733.29
#Sta/Elev= 30
  4323.3  888.33  4417.1  872.11  4520.2  850.49  4548.1  842.06  4561.6  840.38
  4583.0  834.16  4605.4  829.90  4614.6  829.92  4724.1  826.27  4879.1  825.40
  4906.4  823.74  4943.3  826.42  4956.5  825.01  4962.7  822.63  4969.9  823.90
  4991.1  821.70  4992.9  817.70  5007.1  817.70  5008.9  821.70  5017.4  825.20
  5106.3  825.55  5126.4  830.88  5134.7  830.96  5148.0  830.82  5178.9  843.44
  5199.4  846.03  5213.3  850.44  5249.8  855.48  5362.8  868.00  5440.3  873.34
#Mann=9,-1,0
  4323.3    0.14       0  4614.6    0.08       0  4879.1    0.14       0
  4991.1    0.05       0  5008.9    0.14       0  5017.4    0.08       0
  5106.3    0.08       0  5134.7    0.14       0  5249.8    0.08       0
Bank Sta=4991.1,5008.9
XS Rating Curve= 0
Exp/Cntr=0.5,0.3

Type RM Length L Ch R = 1,55830,195,195,195
BEGIN DESCRIPTION:
Union Church Road  FC - us
END DESCRIPTION:
XS GIS Cut Line= 3
      1522884.11       881403.14      1522636.86       880980.55
      1522564.93       880324.19
#Sta/Elev= 30
  4304.9  892.77  4400.9  878.72  4411.5  878.00  4476.0  866.31  4498.4  861.44
  4530.4  856.32  4559.4  849.63  4591.5  844.14  4612.9  838.71  4642.5  833.29
  4656.4  832.30  4793.3  824.98  4857.1  825.40  4939.4  823.84  4953.7  823.29
  4978.0  825.33  4983.5  823.10  4992.5  817.50  5007.5  817.50  5016.5  823.10
  5052.5  823.80  5164.1  825.57  5182.3  826.72  5201.1  836.40  5238.0  839.04
  5294.3  855.00  5348.5  861.52  5392.3  864.87  5433.9  866.72  5454.8  868.93
#Mann=9,-1,0
  4304.9    0.14       0  4656.4    0.08       0  4939.4    0.14       0
  4983.5    0.05       0  5016.5    0.14       0  5052.5    0.08       0
  5164.1    0.14       0  5201.1    0.08       0  5238.0    0.14       0
#XS Ineff=2,0
    0.00 4855.00  833.76 5145.00    0.00  834.56
Permanent Ineff=
       F       F
Bank Sta=4983.5,5016.5
XS Rating Curve= 0
Exp/Cntr=0.5,0.3

Type RM Length L Ch R =3,55726,,,
BEGIN DESCRIPTION:
Union Cross Church Road  FC - TOR
Structure ID: LDS_FC_08
Approximate Survey Structure
END DESCRIPTION:
Bridge Culvert--1,0,-1,-1,0
Deck Dist Width WeirC Skew NumUp NumDn MinLoCord MaxHiCord MaxSubmerge Is_Ogee
86,36,3,,13,13,,,0.95,0,1,1,,,
  4286.3  4482.5  4599.4  4773.9  4906.3  4941.0  4941.0  5059.0  5059.0  5068.7
  5202.8  5302.2  5459.3
  895.81  867.92  855.81  838.11  832.50  832.50  832.50  832.50  832.50  832.50
  838.65  851.91  870.75
  797.50  797.50  797.50  797.50  797.50  797.50  830.20  830.20  797.50  797.50
  797.50  797.50  797.50
  4286.3  4482.5  4599.4  4773.9  4906.3  4941.0  4941.0  5059.0  5059.0  5068.7
  5202.8  5302.2  5459.3
  895.81  867.92  855.81  838.11  832.50  832.50  832.50  832.50  832.50  832.50
  838.65  851.91  870.75
  797.50  797.50  797.50  797.50  797.50  797.50  830.20  830.20  797.50  797.50
  797.50  797.50  797.50
Pier Skew, UpSta & Num, DnSta & Num=,4970.5,2,4970.5,2,0,0,0,0,0
       1       1
  824.85  830.20
       1       1
  824.38  830.20
Pier Skew, UpSta & Num, DnSta & Num=,5029.5,2,5029.5,2,0,0,0,0,0
       1       1
  823.47  830.20
       1       1
  823.31  830.20
Abutment Skew #Up #Dn=,2,2
  4941.0  4957.0
  830.20  823.63
  4941.0  4957.0
  830.20  826.72
Abutment Skew #Up #Dn=,2,2
  5043.0  5059.0
  823.85  830.20
  5043.0  5059.0
  825.63  830.20
BR Coef=1,1,0,1.25,0,,,0.8,0,2,0,
WSPro=,,,, 1 ,,,, 0 ,,,, 0 ,,,,-1 ,-1 ,-1 , 0 , 0 , 0 , 0 , 0
BC Design=,,0,,0,,,,,,

Type RM Length L Ch R = 1,55635,586,586,586
BEGIN DESCRIPTION:
Union Church Road  FC - ds
END DESCRIPTION:
XS GIS Cut Line= 3
      1522969.53       881358.18      1522834.67       880994.04
      1522749.25       880315.21
#Sta/Elev= 30
  4337.5  888.27  4378.1  883.51  4419.7  876.67  4443.7  873.04  4483.8  870.10
  4532.9  864.26  4567.3  860.57  4593.1  851.61  4620.4  844.43  4693.9  831.56
  4761.4  827.69  4824.8  824.53  4871.0  825.24  4921.4  824.73  4957.3  826.73
  4983.5  822.24  4992.5  817.25  5007.5  817.25  5016.5  821.98  5040.3  825.73
  5044.4  825.51  5062.8  823.76  5088.6  823.92  5133.9  827.07  5182.4  833.97
  5210.2  836.04  5227.6  839.28  5252.9  846.64  5311.4  857.01  5410.0  867.32
#Mann=9,-1,0
  4337.5    0.14       0  4419.7    0.08       0  4532.9    0.14       0
  4761.4    0.08       0  4871.0    0.14       0  4983.5    0.05       0
  5016.5    0.14       0  5044.4    0.08       0  5133.9    0.14       0
#XS Ineff=2,0
    0.00 4868.00  833.41 5132.00    0.00  834.05
Permanent Ineff=
       F       F
Bank Sta=4983.5,5016.5
XS Rating Curve= 0
Exp/Cntr=0.5,0.3

Type RM Length L Ch R = 1,55049,961,961,961
BEGIN DESCRIPTION:
Forbush Creek - 55.0
END DESCRIPTION:
XS GIS Cut Line= 2
      1523414.61       881137.91      1523234.77       880085.87
#Sta/Elev= 30
  4466.8  875.35  4498.2  872.58  4516.6  869.25  4537.8  868.00  4578.3  861.60
  4611.7  859.38  4650.2  852.57  4746.4  840.90  4811.3  829.67  4831.0  826.70
  4847.0  823.97  4883.8  821.91  4949.9  824.30  4982.4  821.69  4992.1  818.94
  4993.7  814.94  5006.3  814.94  5007.9  818.94  5016.1  823.49  5021.6  823.57
  5049.2  821.57  5148.2  822.10  5171.8  823.88  5187.6  826.70  5224.5  837.90
  5268.7  845.67  5322.8  851.23  5471.0  859.21  5518.3  863.52  5534.1  866.77
#Mann=7,-1,0
  4466.8    0.14       0  4811.3    0.08       0  4831.0    0.14       0
  4992.1    0.05       0  5007.9    0.14       0  5021.6    0.08       0
  5187.6    0.14       0
Bank Sta=4992.1,5007.9
XS Rating Curve= 0
Exp/Cntr=0.3,0.1

Type RM Length L Ch R = 1,54088,1267,1267,1267
BEGIN DESCRIPTION:
Forbush Creek - 54.0
END DESCRIPTION:
XS GIS Cut Line= 3
      1524556.52       881106.46      1524417.14       880634.39
      1523837.18       879942.02
#Sta/Elev= 30
  4129.8  871.28  4314.3  861.72  4491.2  855.13  4514.1  851.76  4540.3  850.21
  4567.0  845.98  4614.2  837.08  4632.8  832.16  4670.3  827.56  4696.3  826.93
  4716.1  824.58  4759.1  825.76  4778.4  823.39  4876.4  819.93  4941.5  821.05
  4980.2  815.96  4992.1  816.02  4993.7  812.02  5006.3  812.02  5007.9  816.02
  5017.9  821.28  5034.1  820.58  5128.2  819.12  5208.3  820.20  5231.1  821.53
  5251.1  825.79  5312.4  850.52  5337.9  858.39  5371.2  866.20  5525.2  881.67
#Mann=5,-1,0
  4129.8    0.14       0  4992.1    0.05       0  5007.9    0.14       0
  5034.1    0.08       0  5208.3    0.14       0
Bank Sta=4992.1,5007.9
XS Rating Curve= 0
Exp/Cntr=0.3,0.1
