HEC-RAS study North Deep Creek.prj: North Deep Creek Limited Detail Study

--- North Deep Creek.g01 (geometry) --- (continued)

Type RM Length L Ch R = 1 ,51322   ,382,382,382
BEGIN DESCRIPTION:
North Deep Creek 139.0
END DESCRIPTION:
XS GIS Cut Line= 4
      1510784.39       879424.37      1510653.36       879238.17
      1510046.62       879041.67      1509715.62       879020.98
#Sta/Elev= 30
  4688.2  856.11  4693.9  855.07  4798.1  844.75  4867.5  835.16  4897.9  831.43
  4935.6  828.07  4951.5  825.57  4972.3  825.36  4978.3  821.23  4979.8  818.23
  5020.2  818.23  5021.7  821.23    5022  823.68  5035.4  824.29  5049.8  823.42
  5070.6  823.34  5152.1  822.65  5410.5  823.13  5440.1  822.33  5475.1  823.62
  5548.2  823.82  5619.2  826.52    5643  828.66  5682.1   834.9  5763.9  850.61
  5836.6  860.64    5847  861.23  5860.5  863.29  5877.1  863.19  5885.3  863.36
#Mann= 6 ,-1 , 0
  4688.2     .14       0  4978.3    .045       0  5021.7     .14       0
  5070.6     .07       0    5643     .14       0  5877.1     .07       0
#XS Ineff= 2 , 0
       0                  5296.8       0  844.34
Permanent Ineff=
       F       F
Bank Sta=4978.3,5021.7
Exp/Cntr=0.3,0.1

Type RM Length L Ch R = 1 ,50940   ,203,203,203
BEGIN DESCRIPTION:
North Deep Creek 138.0
END DESCRIPTION:
XS GIS Cut Line= 5
      1511011.87       879155.42      1510891.24       879086.48
       1510467.2       878786.56      1510232.78       878627.98
      1510167.28       878490.09
#Sta/Elev= 30
  4446.2  850.14  4501.4  845.45  4518.7  841.85  4531.5  837.92    4537  837.69
    4559  831.38  4582.4  826.89  4620.9  823.94  4673.2  823.19  4754.9  822.73
  4861.6  825.38  4919.2  823.58  4977.2  824.16  4978.3  820.57  4979.8  817.57
  5020.2  817.57  5021.7  820.57  5022.8  821.83  5025.9  823.31  5033.4  823.55
  5042.8  822.35  5064.3  823.28  5095.1  822.58  5136.7  824.45    5251  824.01
  5315.5  825.19  5381.4  830.47  5481.5  843.69  5521.9  851.02  5540.2  853.25
#Mann= 4 ,-1 , 0
  4446.2     .09       0  4673.2     .14       0  4978.3    .045       0
  5021.7     .14       0
#XS Ineff= 2 , 0
       0                  5150.1       0  839.83
Permanent Ineff=
       F       F
Bank Sta=4978.3,5021.7
Exp/Cntr=0.3,0.1

Type RM Length L Ch R = 1 ,50737   ,125,125,125
BEGIN DESCRIPTION:
North Deep Creek 137.0
END DESCRIPTION:
XS GIS Cut Line= 5
      1511061.92       879048.57       1510939.5       879012.36
       1510772.3       878846.89      1510713.69       878790.01
      1510729.21       878658.99
#Sta/Elev= 30
  4555.3  849.55  4581.9  844.57  4634.8  842.34  4648.4   842.1  4659.8  841.08
  4670.6  839.13    4683  833.33  4694.7  829.82  4729.9  823.43  4772.1  822.63
  4785.1  821.97  4808.4  822.65  4829.7  822.22  4834.5  822.77  4846.5  822.64
  4893.5  822.61    4914  823.38  4959.4  823.43  4978.3  820.22  4979.8  817.22
  5020.2  817.22  5021.7  820.22  5053.3  832.77  5062.2  835.66  5065.1  836.28
  5073.4  837.63  5087.4  837.66  5092.6     838  5110.9  840.02  5131.8  841.66
#Mann= 4 ,-1 , 0
  4555.3     .09       0  4846.5     .14       0  4978.3    .045       0
  5021.7     .14       0
Bank Sta=4978.3,5021.7
Exp/Cntr=0.5,0.3

Type RM Length L Ch R = 1 ,50612   ,121,121,121
BEGIN DESCRIPTION:
Country Club Rd (NDC) us
END DESCRIPTION:
XS GIS Cut Line= 5
        1511136.       879024.43      1510972.25       878893.43
      1510856.76       878800.35      1510787.81       878714.16
      1510768.86        878605.6
#Sta/Elev= 30
  4610.5   854.5  4633.8  850.22  4671.3  847.09  4677.9  845.65  4692.9   843.8
  4761.7  841.22  4780.4  840.03  4785.9  839.16  4802.2  838.76    4824   835.9
  4828.5  834.56  4845.9   826.9  4850.9  826.08  4866.2  825.88  4887.1  824.53
  4896.7  824.76  4932.9  824.24  4956.3  822.61  4977.5     824  4988.5     817
  5011.5     817  5022.5     824  5040.1  831.23    5049  832.27  5078.3  838.46
  5083.1  839.06  5138.1  840.44  5157.8  841.47  5181.1  848.81  5189.1  848.86
#Mann= 5 ,-1 , 0
  4610.5     .09       0  4896.7     .14       0  4977.5    .045       0
  5022.5     .14       0  5138.1     .08       0
#XS Ineff= 2 , 0
       0  4922.5   837.8  5077.5       0  838.99
Permanent Ineff=
       F       F
Bank Sta=4977.5,5022.5
Exp/Cntr=0.5,0.3

Type RM Length L Ch R = 3 ,50578   ,,,
BEGIN DESCRIPTION:
Country Club Rd (NDC) tor
Structure ID: LDS_NDC_10
Approximate Survey Structure
END DESCRIPTION:
Bridge Culvert--1,0,-1,-1, 0
Deck Dist Width WeirC Skew NumUp NumDn MinLoCord MaxHiCord MaxSubmerge Is_Ogee
20,28,3,0, 7, 7, , , 0.95, 0, 1,1,,
    4737  4828.8  4942.5  4942.5  5057.5  5057.5  5081.1
  841.47   837.8   837.8   837.8   837.8   837.8   837.8
  796.99  796.99  796.99   834.3   834.3  796.99  796.99
    4737  4828.8  4942.5  4942.5  5057.5  5057.5  5081.1
  841.47   837.8   837.8   837.8   837.8   837.8   837.8
  796.99  796.99  796.99   834.3   834.3  796.99  796.99
Pier Skew, UpSta & Num, DnSta & Num=  ,4971.3, 2 ,4971.3, 2 , 0 , 0 , 0 ,0,0
     1.7     1.7
  823.31   834.3
     1.7     1.7
  823.61   834.3
Pier Skew, UpSta & Num, DnSta & Num=  ,5028.8, 2 ,5028.8, 2 , 0 , 0 , 0 ,0,0
     1.7     1.7
  826.53   834.3
     1.7     1.7
  824.08   834.3
Abutment Skew #Up #Dn= , 2 , 2
  4942.5  4962.8
   834.3  822.99
  4942.5  4962.8
   834.3  823.79
Abutment Skew #Up #Dn= , 2 , 2
  5037.3  5057.5
  830.04   834.3
  5037.3  5057.5
  824.51   834.3
BR Coef= 1 , 1 , 0 ,1.25, 0 ,,,0.8,-1,2,0,
WSPro=,,,, 1 ,,,, 0 ,,,, 0 ,,,,-1 ,-1 ,-1 , 0 , 0 , 0 , 0 , 0
BC Design=,, 0 ,, 0 ,,,,,,
BC HTab HWMax=854.5

Type RM Length L Ch R = 1 ,50491   ,71,71,71
BEGIN DESCRIPTION:
Country Club Rd (NDC) ds
END DESCRIPTION:
XS GIS Cut Line= 4
       1511203.2       878943.38      1511029.13       878755.53
      1510892.96       878676.24      1510805.02        878602.1
#Sta/Elev= 30
  4626.5  847.09  4641.2  846.88  4658.2   845.1  4699.3  844.76  4722.9  843.28
  4751.2   840.3  4788.5  838.47    4832  830.96  4862.8   826.8  4874.3  825.31
    4901  823.57  4920.1  823.02  4955.8  823.21  4960.2  823.87  4969.9  823.58
  4977.5  823.96  4988.5  816.96  5011.5  816.96  5022.5  823.96  5037.8  824.54
  5042.2  825.35  5046.4  825.44  5049.2  827.83  5057.9  831.65  5066.7   834.4
  5072.4  838.23  5104.7  844.94  5114.2  847.46  5135.1  850.52  5155.2  851.41
#Mann= 5 ,-1 , 0
  4626.5     .09       0  4862.8     .14       0  4977.5    .045       0
  5022.5     .14       0  5104.7     .08       0
#XS Ineff= 2 , 0
       0  4869.5   837.8  5130.5       0     841
Permanent Ineff=
       F       F
Bank Sta=4977.5,5022.5
Exp/Cntr=0.5,0.3

Type RM Length L Ch R = 1 ,50420   ,328,328,328
BEGIN DESCRIPTION:
North Deep Creek 136.0
END DESCRIPTION:
XS GIS Cut Line= 4
      1511191.26       878801.07      1511025.52       878685.44
      1510948.44       878623.78      1510782.77       878577.54
#Sta/Elev= 30
  4734.9  840.65  4758.4  839.19  4774.2  838.93  4790.2  837.85  4839.1  833.52
  4846.8  832.32  4876.9  827.93  4891.9  824.78  4903.4  823.19  4919.1   822.2
  4924.8  821.49  4946.2  824.14  4985.8  821.42    4987  819.93  4987.9  816.93
  5012.1  816.93    5013  819.93  5013.4  823.71  5046.8  831.48  5066.8  837.43
  5077.2  839.48  5116.4  844.75    5121  845.47  5123.7  846.29  5147.3  848.93
  5164.4  851.49  5169.6  851.86  5189.6  852.18  5196.3  851.89  5207.7   850.8
#Mann= 5 ,-1 , 0
  4734.9     .09       0  4846.8     .14       0    4987    .045       0
    5013     .14       0  5116.4     .08       0
Bank Sta=4987,5013
Exp/Cntr=0.3,0.1

Type RM Length L Ch R = 1 ,50092   ,368,368,368
BEGIN DESCRIPTION:
North Deep Creek 135.0
END DESCRIPTION:
XS GIS Cut Line= 4
      1511322.27       878727.85      1511237.48       878558.26
      1511156.55       878327.03      1511087.17        878203.7
#Sta/Elev= 30
  4717.5  837.78  4736.9  838.17  4752.9  837.81  4799.2  834.95  4852.7  829.84
  4868.3  828.82  4892.2  826.07  4916.7  823.98  4950.4  821.38  4972.1  820.82
  4982.6  819.81  4983.8  816.81  5016.2  816.81  5017.4  819.81  5021.7  823.77
  5029.1  824.46  5051.4  824.95  5060.6  825.59  5122.8  822.17  5154.4  821.72
  5193.8  823.08  5204.5  828.25  5214.4  831.17  5229.9  838.99  5241.2  846.15
  5245.2  847.88    5257  850.65    5284  854.08  5286.7  854.03  5293.6  854.14
#Mann= 5 ,-1 , 0
  4717.5     .09       0  4799.2     .14       0  4982.6    .045       0
  5017.4     .14       0  5286.7     .08       0
#XS Ineff= 2 , 0
       0                    5120       0     838
Permanent Ineff=
       F       F
Bank Sta=4982.6,5017.4
Exp/Cntr=0.3,0.1

Type RM Length L Ch R = 1 ,49724   ,179,179,179
BEGIN DESCRIPTION:
North Deep Creek 134.0
END DESCRIPTION:
XS GIS Cut Line= 4
       1511561.2       878666.18       1511561.2       878515.87
      1511534.22       878330.89      1511437.88       878172.89
#Sta/Elev= 30
  4732.8  838.92  4745.7  838.74  4764.2  839.44  4776.3  839.04  4780.3  838.43
  4820.5  836.17  4825.7   835.7  4859.7  829.53  4879.7  827.17  4900.4   823.5
  4914.2     822    4943  821.75  4981.9  823.34  4984.2  822.67  4984.8  819.36
  4985.9  816.36  5014.1  816.36  5015.2  819.36    5022  821.91  5029.6  822.76
  5050.8  824.43  5067.9  824.23  5091.2  826.16  5098.1  827.93  5113.2  832.84
  5119.9  834.43    5144  835.72  5183.7  838.49  5220.1  839.99  5255.1  840.56
#Mann= 4 ,-1 , 0
  4732.8     .14       0  4984.8    .045       0  5015.2     .14       0
    5144     .08       0
Bank Sta=4984.8,5015.2
Exp/Cntr=0.3,0.1

Type RM Length L Ch R = 1 ,49545   ,365,365,365
BEGIN DESCRIPTION:
North Deep Creek 133.0
END DESCRIPTION:
XS GIS Cut Line= 4
      1511923.47       878411.82      1511780.87       878357.86
      1511615.15       878280.79      1511495.69       878184.45
#Sta/Elev= 30
  4749.4  855.15  4768.3  852.63  4811.2   848.4  4813.4  848.49  4842.5  843.43
  4845.5  843.77  4853.1  842.22  4860.7  839.33  4880.6  835.04  4890.2  834.08
  4896.8  832.87  4908.9  829.21  4924.6  825.73  4949.7   822.5  4969.8  822.69
  4981.8  819.11    4983  816.11    5017  816.11  5018.2  819.11  5050.6  823.18
  5064.1  822.41  5099.4     822  5119.3  823.82  5135.8  827.49  5147.3  833.27
  5154.3  834.93  5171.3  836.61  5212.4  839.65  5232.9  840.52  5238.1  840.36
#Mann= 4 ,-1 , 0
  4749.4     .14       0  4981.8    .045       0  5018.2     .14       0
  5171.3     .08       0
Bank Sta=4981.8,5018.2
Exp/Cntr=0.3,0.1

Type RM Length L Ch R = 1 ,49180   ,331,331,331
BEGIN DESCRIPTION:
North Deep Creek 131.0
END DESCRIPTION:
XS GIS Cut Line= 4
      1512046.82       878169.06      1511927.32       878061.12
      1511827.12       877980.19      1511595.86       878034.15
#Sta/Elev= 30
  4790.4  853.78  4864.4  842.09  4877.4  839.36  4897.9  835.43  4945.3  824.72
  4952.4  823.64  4968.3  822.11  4969.6  822.19  4979.5  818.42  4980.8  815.42
  5019.2  815.42  5020.5  818.42  5033.6  825.15  5036.1  824.91  5055.4  824.13
  5059.1  824.24  5069.6   823.4  5076.6  823.27  5080.2  822.52  5092.4  822.13
  5099.1  821.68  5123.7  825.23  5136.6   828.3  5152.4  829.47  5162.9  829.95
  5186.8  832.02  5224.6  834.37  5285.9     837  5297.5  837.78  5317.7  838.52
#Mann= 4 ,-1 , 0
  4790.4     .14       0  4979.5    .045       0  5020.5     .14       0
  5152.4     .08       0
Bank Sta=4979.5,5020.5
Exp/Cntr=0.3,0.1

Type RM Length L Ch R = 1 ,48849   ,315,315,315
BEGIN DESCRIPTION:
North Deep Creek 130.0
END DESCRIPTION:
XS GIS Cut Line= 5
      1512239.48       878061.13      1512143.13       877864.57
      1511896.48       877656.47      1511669.11       877517.73
      1511599.73       877355.84
#Sta/Elev= 30
  4555.1  853.18  4580.4  850.03  4670.1  841.71  4724.8  837.15  4744.3  834.99
  4761.6  830.54  4787.4  825.27    4812  822.47  4865.2  823.04  4938.2  822.81
  4981.8  818.05    4983  815.05    5017  815.05  5018.2  818.05  5023.4  822.24
  5070.7  822.04  5082.1  821.57  5095.4  821.83  5101.3  821.35  5148.8  826.32
  5221.6  832.83  5244.1  833.96    5284   834.8  5344.3  837.73  5363.1  839.05
  5379.2  841.39  5454.9  845.25  5515.7  849.39  5521.7  850.25  5539.2  851.87
#Mann= 4 ,-1 , 0
  4555.1     .14       0  4981.8    .045       0  5018.2     .14       0
  5521.7     .08       0
Bank Sta=4981.8,5018.2
Exp/Cntr=0.3,0.1

Type RM Length L Ch R = 1 ,48534   ,432,432,432
BEGIN DESCRIPTION:
North Deep Creek 129.0
END DESCRIPTION:
XS GIS Cut Line= 5
      1512555.51        877872.3      1512266.45       877648.76
      1512143.13        877486.9      1512139.28       877359.72
      1512135.42       877147.79
#Sta/Elev= 30
  4433.5  847.53  4459.8  845.09  4487.5  846.23  4549.4  842.24  4630.8  838.47
  4672.8  838.07  4696.9  835.59  4713.7  834.25  4720.7  834.18  4748.4  831.68
  4802.8  829.69  4855.2  822.69  4911.1     822  4947.1  822.05  4967.9  822.71
  4981.8  816.89    4983  813.89    5017  813.89  5018.2  816.89  5021.6  820.23
  5030.9  821.99  5041.9   822.3  5068.7  824.48  5090.1  825.57    5105  827.56
  5150.1  831.71  5234.6  835.43  5260.6  837.42  5290.3  841.74  5341.6  847.04
#Mann= 3 ,-1 , 0
  4433.5     .14       0  4981.8    .045       0  5018.2     .14       0
Bank Sta=4981.8,5018.2
Exp/Cntr=0.3,0.1

Type RM Length L Ch R = 1 ,48102   ,340,340,340
BEGIN DESCRIPTION:
North Deep Creek 128.0
END DESCRIPTION:
XS GIS Cut Line= 4
      1512698.05       877525.42      1512574.76       877440.65
      1512486.12       877271.08      1512277.97       877182.43
#Sta/Elev= 30
  4734.3   848.3  4745.5  846.35  4753.1  846.44  4775.2  844.17  4795.8  840.36
  4833.5  836.31  4866.9  829.33    4879  825.87  4893.7  823.35  4902.1  820.84
  4934.4  820.65  4958.3  822.49  4963.2  822.24  4981.8  815.13    4983  812.13
    5017  812.13  5018.2  815.13  5018.5  820.49  5025.7  823.05  5057.4  822.93
  5070.1  821.98  5119.9   822.2  5127.8  822.87    5144  825.35  5165.9  829.36
  5181.3  830.64  5210.7  834.84  5253.4  839.35  5274.9  842.18  5301.5  844.13
#Mann= 3 ,-1 , 0
  4734.3     .14       0  4981.8    .045       0  5018.2     .14       0
Bank Sta=4981.8,5018.2
Exp/Cntr=0.3,0.1

Type RM Length L Ch R = 1 ,47762   ,388,388,388
BEGIN DESCRIPTION:
North Deep Creek 127.0
END DESCRIPTION:
XS GIS Cut Line= 6
      1512998.71        877355.9       1512863.8       877213.28
      1512748.18       877105.37       1512671.1       877078.39
      1512443.73       877089.95      1512204.81       877120.78
#Sta/Elev= 30
  4621.2  861.44  4637.9   857.7  4700.1   854.9  4726.3  850.89  4783.5   839.3
  4803.6  831.89  4844.9  821.46  4877.2  819.22  4926.2  821.88  4975.7  817.84
    4979  817.38  4981.8  814.76    4983  811.76    5017  811.76  5018.2  814.76
  5019.9  820.06  5025.6   821.9  5031.6  822.28  5063.4  821.93  5088.7  820.37
    5128  821.77  5215.9   821.9  5286.3  824.01  5295.2  823.65  5339.5  827.22
  5363.4     830  5417.4  838.84  5454.9  843.55  5498.2  846.85  5525.9  847.89
#Mann= 3 ,-1 , 0
  4621.2     .14       0  4981.8    .045       0  5018.2     .14       0
Bank Sta=4981.8,5018.2
Exp/Cntr=0.3,0.1

Type RM Length L Ch R = 1 ,47374   ,287,287,287
BEGIN DESCRIPTION:
North Deep Creek 126.0
END DESCRIPTION:
XS GIS Cut Line= 4
      1513033.34        876735.4      1512844.53       876754.67
      1512328.11       876955.07      1512166.24       876955.07
#Sta/Elev= 30
    4837  863.45  4847.6  862.79  4863.8  859.44  4912.3  847.07  4922.1  843.45
  4929.5  838.69  4935.7     836  4975.4  814.53  4981.5  814.21  4982.7  811.21
  5017.3  811.21  5018.5  814.21  5019.2  822.48  5023.5  822.62  5065.4  820.77
    5165  820.21  5185.6  819.12  5196.2  820.02  5262.1  820.36  5290.8  822.22
  5350.6  822.42    5399   820.5  5512.7  821.71    5556  822.84  5575.9  823.81
  5594.7   826.8  5628.1  830.19  5673.5  838.57    5725  844.24  5742.6  849.01
#Mann= 3 ,-1 , 0
    4837     .14       0  4981.5    .045       0  5018.5     .14       0
Bank Sta=4981.5,5018.5
Exp/Cntr=0.3,0.1

Type RM Length L Ch R = 1 ,47087   ,595,595,595
BEGIN DESCRIPTION:
North Deep Creek 125.0
END DESCRIPTION:
XS GIS Cut Line= 5
      1512983.27       876639.06      1512782.87       876554.27
      1512543.93       876604.37      1512293.43       876600.52
      1512154.66       876635.21
#Sta/Elev= 30
  4646.7  861.66    4676  860.35  4718.9  856.87  4758.1  851.17  4782.8  845.14
  4798.7  842.33  4847.5  829.91  4877.7  823.52  4894.1  821.12  4960.8   814.7
  4981.2     815  4983.8  814.11  4984.9  811.11  5015.1  811.11  5016.2  814.11
    5022  821.39  5042.1  821.96  5070.9  819.95  5080.4  818.36  5194.9  821.44
  5230.3  820.52  5249.7  821.77  5260.6   820.8  5289.4  821.63  5328.2  820.19
  5358.1  822.74  5365.5  823.88  5402.5  833.28    5472   853.1    5502  858.15
#Mann= 3 ,-1 , 0
  4646.7     .14       0  4983.8    .045       0  5016.2     .14       0
Bank Sta=4983.8,5016.2
Exp/Cntr=0.3,0.1

Type RM Length L Ch R = 1 ,46492   ,524,524,524
BEGIN DESCRIPTION:
North Deep Creek 124.0
END DESCRIPTION:
XS GIS Cut Line= 3
      1512948.58       876600.52      1512455.29       876114.93
      1512385.91       876033.99
#Sta/Elev= 30
  4283.4  857.97  4319.3  853.65    4335  850.81  4358.9  845.79  4430.2  828.01
  4440.6  825.81  4457.9  823.53  4482.1  823.02  4503.8  820.95  4591.5  819.74
  4628.9  820.87    4671  819.35  4701.6  821.68  4730.1  820.41  4743.7  821.22
  4775.7  821.49  4817.1   821.1  4888.8  818.17  4921.1  816.09  4943.7  815.53
  4962.6  814.03  4978.6     814  4981.5  813.23  4982.7  810.23  5017.3  810.23
  5018.5  813.23  5020.3   820.1  5052.1  842.78  5072.1  857.85  5082.2  862.13
#Mann= 3 ,-1 , 0
  4283.4     .14       0  4981.5    .045       0  5018.5     .14       0
Bank Sta=4981.5,5018.5
Exp/Cntr=0.3,0.1

Type RM Length L Ch R = 1 ,45968   ,209,209,209
BEGIN DESCRIPTION:
North Deep Creek 123.0
END DESCRIPTION:
XS GIS Cut Line= 5
      1512975.56       876615.95      1512987.12       876338.46
      1512929.31       876022.44      1512898.48       875918.39
      1512790.57       875798.92
#Sta/Elev= 30
  4320.6   860.3  4358.3  855.54  4365.9  855.31  4389.9  850.33  4425.1  844.62
  4465.5  840.31  4545.1  827.71  4572.1  824.39  4679.8  819.09  4746.9  817.95
  4783.8  818.48  4859.4   817.7  4946.2  819.24  4973.8  814.79  4982.5  815.03
  4983.8   812.9  4984.9   809.9  5015.1   809.9  5016.2   812.9  5018.1  816.24
  5050.7  819.93  5101.1  818.48  5111.4  820.86  5124.1  826.34  5128.9  827.02
  5136.8  831.21  5142.2  835.75  5151.9  839.15  5161.9  842.19  5189.1   848.1
#Mann= 3 ,-1 , 0
  4320.6     .14       0  4983.8    .045       0  5016.2     .14       0
Bank Sta=4983.8,5016.2
Exp/Cntr=0.3,0.1

Type RM Length L Ch R = 1 ,45759   ,339,339,339
BEGIN DESCRIPTION:
North Deep Creek 122.0
END DESCRIPTION:
XS GIS Cut Line= 4
      1512994.83       876619.79      1513006.39       876338.46
      1513041.07        875883.7      1513029.51       875741.11
#Sta/Elev= 30
  4190.3  860.42  4229.7  856.25    4268  850.63  4283.5  847.35  4307.9  845.35
  4417.4  829.31  4457.6  824.68  4498.1  823.91    4573  819.43  4580.7  818.42
    4596  818.62  4618.6  817.24  4705.1  818.45  4778.6  817.57  4840.7  819.42
  4882.7  817.88  4900.6  818.93  4939.5  817.91  4954.3  818.63    4960   818.5
  4973.7  814.21  4983.8  812.86  4984.9  809.86  5015.1  809.86  5016.2  812.86
  5018.4  823.92  5040.4  840.94  5047.8  843.38  5062.7  845.23    5071  848.22
#Mann= 3 ,-1 , 0
  4190.3     .14       0  4983.8    .045       0  5016.2     .14       0
Bank Sta=4983.8,5016.2
Exp/Cntr=0.3,0.1

Type RM Length L Ch R = 1 ,45420   ,306,306,306
BEGIN DESCRIPTION:
North Deep Creek 121.0
END DESCRIPTION:
XS GIS Cut Line= 5
      1513025.66       876604.38      1513029.51       876373.14
      1513125.86       876130.35      1513187.52       876010.88
      1513264.58        875852.9
#Sta/Elev= 30
  4458.3  858.78    4567  845.81  4625.3  837.53  4654.8     832  4699.9  827.61
  4713.8  825.23    4732  824.41  4778.6  819.17  4831.8  817.26  4880.5   817.7
    4936  817.18  4972.2  818.45  4978.5  817.19  4981.5  812.41  4982.7  809.41
  5017.3  809.41  5018.5  812.41  5021.2  814.04  5039.6  818.61  5049.3  819.47
  5076.6  819.56    5095  818.61  5107.7   819.4  5131.2  818.39  5143.5  819.44
  5166.9   830.8  5183.2   840.3  5199.8  848.52  5227.9  855.19    5261  858.83
#Mann= 3 ,-1 , 0
  4458.3     .14       0  4981.5    .045       0  5018.5     .14       0
Bank Sta=4981.5,5018.5
Exp/Cntr=0.3,0.1

Type RM Length L Ch R = 1 ,45114   ,461,461,461
BEGIN DESCRIPTION:
North Deep Creek 120.0
END DESCRIPTION:
XS GIS Cut Line= 4
      1513272.31       876639.04      1513337.82       876508.03
      1513407.19        876026.3      1513457.31       875941.48
#Sta/Elev= 30
  4346.5  854.48  4389.3  849.79  4434.3  843.42    4476   834.2  4490.1  830.39
  4518.5  820.31  4529.1  817.53  4546.2  817.48  4564.3  816.41  4603.4  817.01
  4616.4  817.74  4627.9  816.82    4685  817.84  4752.4  816.72  4787.6  816.97
  4823.7   816.3  4862.1  817.04  4900.3  818.41  4945.1  817.96  4957.1  818.87
    4976  818.41  4979.7  817.73  4981.5  811.27  4982.7  808.27  5017.3  808.27
  5018.5  811.27  5027.8  812.94    5034  815.86  5067.5  836.44  5078.2  840.44
#Mann= 3 ,-1 , 0
  4346.5     .14       0  4981.5    .045       0  5018.5     .14       0
Bank Sta=4981.5,5018.5
Exp/Cntr=0.3,0.1

Type RM Length L Ch R = 1 ,44653   ,225,225,225
BEGIN DESCRIPTION:
North Deep Creek 119.0
END DESCRIPTION:
XS GIS Cut Line= 5
      1513584.45       876654.52      1513657.69       876430.95
      1513676.95        876284.5      1513669.25       876095.67
      1513615.28       875945.32
#Sta/Elev= 30
  4696.5  836.62  4739.1  832.18  4793.8  827.91  4827.5  826.26  4842.3  826.22
    4940  815.76    4954  815.93  4967.8  817.91  4970.8  816.61  4976.9  810.63
  4978.4  807.63  5021.6  807.63  5023.1  810.63    5027  815.51  5033.5  817.67
  5037.5  818.14  5065.1  818.61  5091.8  817.31  5106.7  818.41  5135.5  817.33
  5178.3  817.97  5191.2   816.9  5204.8  817.17  5229.2  816.48  5265.7  817.73
  5286.8  819.75  5353.8  830.25    5366   830.9  5401.9  835.65  5428.2   836.6
#Mann= 3 ,-1 , 0
  4696.5     .14       0  4976.9    .045       0  5023.1     .14       0
Bank Sta=4976.9,5023.1
Exp/Cntr=0.3,0.1

Type RM Length L Ch R = 1 ,44428   ,238,238,238
BEGIN DESCRIPTION:
North Deep Creek 118.0
END DESCRIPTION:
XS GIS Cut Line= 4
      1513842.67       876623.66      1513815.69       876423.24
      1513777.15       876080.25      1513653.83       875941.51
#Sta/Elev= 30
  4845.8  846.24  4885.2  841.06  4921.4  834.67  4959.5  826.81  4977.5  820.01
  4981.5  810.34  4982.7  807.34  5017.3  807.34  5018.5  810.34  5021.3  813.75
  5041.7  814.01  5055.8  811.97  5064.7   811.4  5077.1  812.51  5084.5  812.46
  5099.6  816.33  5114.9  817.34  5143.6  817.24  5154.7  816.52  5181.1  817.29
  5299.5  816.49  5328.9   817.7    5366  816.32  5403.2  817.14  5414.6   816.6
  5495.6  828.44  5518.2  830.91  5548.1  835.43  5556.3  834.79  5578.8  836.12
#Mann= 3 ,-1 , 0
  4845.8     .14       0  4981.5    .045       0  5018.5     .14       0
Bank Sta=4981.5,5018.5
Exp/Cntr=0.3,0.1

Type RM Length L Ch R = 1 ,44190   ,192,192,192
BEGIN DESCRIPTION:
North Deep Creek 117.0
END DESCRIPTION:
XS GIS Cut Line= 5
      1514073.91       876334.61      1513965.99       876272.94
      1513877.35       876261.38      1513788.72       876060.98
      1513661.54       875929.96
#Sta/Elev= 30
  4818.7  842.92  4863.8  841.24  4885.6  839.24  4896.8  835.89  4918.3  830.39
  4955.5  818.64  4962.2  816.85  4975.8  814.78  4976.9  809.59  4978.4  806.59
  5021.6  806.59  5023.1  809.59    5025  816.99  5030.9  817.77  5040.9  817.51
  5048.5  816.62  5070.4  817.05  5090.1   816.5  5114.3  816.65    5136  815.84
  5179.9  817.43  5223.6  816.03    5268  816.54  5288.3  819.47  5301.5  822.13
  5313.3  823.61  5338.1  827.82  5406.5  835.46  5409.2  835.24  5434.1  836.17
#Mann= 3 ,-1 , 0
  4818.7     .14       0  4976.9    .045       0  5023.1     .14       0
Bank Sta=4976.9,5023.1
Exp/Cntr=0.3,0.1

Type RM Length L Ch R = 1 ,43998   ,354,354,354
BEGIN DESCRIPTION:
North Deep Creek 116.0
END DESCRIPTION:
XS GIS Cut Line= 4
      1514108.59       876265.24      1514043.07       876114.93
      1513804.13       876030.15      1513669.29       875914.57
#Sta/Elev= 30
  4723.3  837.92  4759.4  836.03  4781.4  833.05  4809.1  831.96  4825.4  829.88
  4843.8  830.33  4857.7  829.09    4881  828.97  4898.7  827.33  4918.9  823.14
  4946.8  816.47  4958.9  815.37  4968.8   815.6  4976.9  809.26  4978.4  806.26
  5021.6  806.26  5023.1  809.26  5024.9  816.38    5045  815.36  5069.7  816.68
  5091.8  815.48  5113.7  815.27  5147.1  816.52  5168.7  819.95  5220.2  827.12
  5234.3  829.69  5259.4  831.91  5277.6   834.4  5292.7  835.34  5318.4   835.9
#Mann= 3 ,-1 , 0
  4723.3     .14       0  4976.9    .045       0  5023.1     .14       0
Bank Sta=4976.9,5023.1
Exp/Cntr=0.3,0.1

Type RM Length L Ch R = 1 ,43644   ,365,365,365
BEGIN DESCRIPTION:
North Deep Creek 115.0
END DESCRIPTION:
XS GIS Cut Line= 4
      1514370.67       875972.38      1514251.18       875787.36
      1513881.21       875706.43      1513557.54       875737.25
#Sta/Elev= 30
  4517.7  839.49  4544.9  837.63  4558.2  835.07  4583.6   832.7  4603.4   829.1
  4629.3  826.79  4647.9     826  4784.4   815.5  4811.2  814.84  4938.8  816.26
  4941.2  816.26    4950  818.43  4967.6  820.37  4975.4  819.14  4976.9   809.2
  4978.4   806.2  5021.6   806.2  5023.1   809.2  5023.9  815.67  5042.3  816.41
  5058.4  815.23    5092  815.18  5114.8  816.93  5131.6  816.48  5147.2  817.14
  5194.2  821.25  5237.9  826.32  5360.3  830.24  5413.3  834.57  5441.8  838.35
#Mann= 5 ,-1 , 0
  4517.7     .14       0  4647.9     .07       0  4938.8     .14       0
  4976.9    .045       0  5023.1     .14       0
Bank Sta=4976.9,5023.1
Exp/Cntr=0.3,0.1

Type RM Length L Ch R = 1 ,43279   ,375,375,375
BEGIN DESCRIPTION:
North Deep Creek 114.0
END DESCRIPTION:
XS GIS Cut Line= 5
      1514424.62       875976.23      1514316.69       875791.21
      1514185.66       875479.05      1514139.41       875286.36
      1514143.27         875086.
#Sta/Elev= 30
  4556.2  844.66  4602.7  840.64  4716.6  825.68    4761  820.94  4853.9  814.56
  4908.8  814.17  4942.1  815.27  4956.1  815.94  4961.2  815.39    4981     809
  4982.2     806  5017.8     806    5019     809  5031.1  814.59  5038.9  816.19
  5066.3  817.11  5117.5  817.28  5172.3  815.05  5226.2  815.11  5266.6  813.42
  5355.4  814.61  5374.2  813.55  5378.6  814.36    5391  814.27  5412.5  827.33
  5430.3  840.66  5446.5  849.56  5457.1  853.51  5468.3   856.3  5507.5  859.47
#Mann= 5 ,-1 , 0
  4556.2     .14       0  4716.6     .07       0  4942.1     .14       0
    4981    .045       0    5019     .14       0
#XS Ineff= 2 , 0
       0  4813.6  838.99  5229.3       0  838.99
Permanent Ineff=
       F       F
Bank Sta=4981,5019
Exp/Cntr=0.3,0.1

Type RM Length L Ch R = 1 ,42904   ,326,326,326
BEGIN DESCRIPTION:
North Deep Creek 113.0
END DESCRIPTION:
XS GIS Cut Line= 4
      1514678.96       875841.34      1514655.83       875706.43
      1514497.82       875355.73      1514305.13       875112.93
#Sta/Elev= 30
  4422.6   851.5  4502.2   836.3  4514.2  833.04  4551.6  820.28  4574.6  815.71
  4600.7  813.77  4632.3  813.18  4663.1   814.4  4726.5  813.01  4767.2  814.25
  4820.8  813.18    4836  814.13  4909.6  813.68  4943.9  815.44    4963  814.97
    4981  808.23  4982.2  805.23  5017.8  805.23    5019  808.23  5022.7  813.65
  5027.8  814.33  5039.8  813.44  5048.8  815.26  5080.7  826.84  5120.2  837.05
  5146.6   842.7  5198.5     852  5240.5   857.7  5246.9  859.64  5254.1  860.51
#Mann= 5 ,-1 , 0
  4422.6     .14       0  4767.2     .07       0  4943.9     .14       0
    4981    .045       0    5019     .14       0
#XS Ineff= 2 , 0
       0  4726.1  838.76               0
Permanent Ineff=
       F       F
Bank Sta=4981,5019
Exp/Cntr=0.3,0.1

Type RM Length L Ch R = 1 ,42578   ,326,326,326
BEGIN DESCRIPTION:
North Deep Creek 112.0
END DESCRIPTION:
XS GIS Cut Line= 4
      1515218.45       874993.47      1514910.18       875012.74
      1514547.92       875078.25      1514312.83       875032.01
#Sta/Elev= 30
    4424  837.05  4463.2   834.3  4473.6  832.57  4503.2  829.99  4540.6  827.79
  4572.8  826.73  4617.2  827.75  4660.3  821.04  4737.8   811.9  4790.7  813.17
  4868.1  813.37  4902.1  811.81  4928.7  813.85  4977.7  815.76    4981  808.04
  4982.2  805.04  5017.8  805.04    5019  808.04  5025.5   814.3  5057.2  813.12
    5100  814.68  5202.1  812.89  5225.1  813.74    5240  822.16  5256.1  837.34
  5266.4  845.75  5284.3  856.38  5294.7  858.13  5309.3  864.72  5340.6  867.28
#Mann= 3 ,-1 , 0
    4424     .14       0    4981    .045       0    5019     .14       0
Bank Sta=4981,5019
Exp/Cntr=0.3,0.1

Type RM Length L Ch R = 1 ,42252   ,427,427,427
BEGIN DESCRIPTION:
North Deep Creek 111.0
END DESCRIPTION:
XS GIS Cut Line= 4
      1515176.05       874939.51      1514906.33       874912.54
      1514594.17       874796.92      1514389.93       874777.66
#Sta/Elev= 30
    4442  835.53  4465.9  834.58  4502.4  831.27  4547.6  830.15  4569.5  828.32
  4598.5  828.16  4641.6  826.06  4690.8  816.76  4739.3  813.02    4762  812.42
  4791.6  812.91  4856.1  811.83  4884.5   813.6  4939.1  814.36    4968  811.43
  4978.7  807.85    4980  804.85    5020  804.85  5021.3  807.85  5022.2  814.45
  5074.2  813.11    5093  816.26    5114  827.42  5138.9  836.72  5164.2  843.57
  5171.1  843.98  5191.7  847.81  5217.8   855.7  5227.5  857.27  5251.1  862.84
#Mann= 3 ,-1 , 0
    4442     .14       0  4978.7    .045       0  5021.3     .14       0
Bank Sta=4978.7,5021.3
Exp/Cntr=0.3,0.1

Type RM Length L Ch R = 1 ,41825   ,251,251,251
BEGIN DESCRIPTION:
North Deep Creek 110.0
END DESCRIPTION:
XS GIS Cut Line= 4
       1515214.6       874893.25      1514994.97       874762.24
       1514682.8       874500.18      1514440.01       874388.42
#Sta/Elev= 30
  4428.3  840.49    4496   834.3  4552.9  828.15  4569.2  825.41  4601.2  822.64
    4623  822.15  4657.7   817.4  4709.3  813.26  4736.8  812.25  4792.9  813.44
  4827.1  811.15  4846.3  812.55  4904.6  812.29    4944   813.7  4950.3  813.14
  4976.3  806.75  4977.8  803.75  5022.2  803.75  5023.7  806.75  5029.1  813.67
  5068.7  811.23  5086.3  812.97  5117.7  811.41  5148.4  813.87  5195.2  814.04
  5235.3   836.3  5264.6  847.75  5300.2  855.85    5343  861.28  5358.9  865.74
#Mann= 3 ,-1 , 0
  4428.3     .14       0  4976.3    .045       0  5023.7     .14       0
Bank Sta=4976.3,5023.7
Exp/Cntr=0.3,0.1

Type RM Length L Ch R = 1 ,41574   ,349,349,349
BEGIN DESCRIPTION:
North Deep Creek 109.0
END DESCRIPTION:
XS GIS Cut Line= 4
      1515191.54       874839.35      1515052.77       874681.31
      1514809.98       874338.32      1514709.78       874230.41
#Sta/Elev= 30
  4352.1   836.4  4374.1  834.31  4427.5  826.55  4457.9  823.28  4595.8  814.69
  4628.7  811.54  4655.7  811.36  4672.4  811.81  4684.5  810.76  4732.6  812.08
  4759.8  811.65  4831.8  812.01  4858.2  812.77    4879  812.52  4895.7  813.59
  4933.4  812.93  4957.7  813.69  4964.5  812.82  4976.3  806.42  4977.8  803.42
  5022.2  803.42  5023.7  806.42  5035.9  814.22  5040.7  814.59  5054.6  817.72
  5068.9   822.4  5083.8  825.62  5102.3  829.17  5125.3  833.03  5129.9  834.48
#Mann= 3 ,-1 , 0
  4352.1     .14       0  4976.3    .045       0  5023.7     .14       0
Bank Sta=4976.3,5023.7
Exp/Cntr=0.3,0.1

Type RM Length L Ch R = 1 ,41225   ,377,377,377
BEGIN DESCRIPTION:
North Deep Creek 108.0
END DESCRIPTION:
XS GIS Cut Line= 4
      1515199.23       874850.92      1515137.56       874638.92
      1515122.14       874376.86      1515137.55       874265.12
#Sta/Elev= 30
  4481.7  838.06  4517.1  834.89    4547  831.01  4575.4  828.44  4598.1  824.51
  4644.5  818.84  4689.4  815.28    4714  814.77  4734.4  813.75    4759  811.33
  4782.9  812.81  4802.3  811.95  4817.2  810.31  4828.5   811.5  4841.4  812.18
  4893.8  813.83  4894.8  813.36  4928.5  810.64  4933.4  810.63    4947  807.71
    4965  807.48  4978.7  806.05    4980  803.05    5020  803.05  5021.3  806.05
  5022.3  812.81  5042.7   830.7  5051.8  836.82  5075.5  845.81  5077.8  846.33
#Mann= 3 ,-1 , 0
  4481.7     .14       0  4978.7    .045       0  5021.3     .14       0
Bank Sta=4978.7,5021.3
Exp/Cntr=0.3,0.1

Type RM Length L Ch R = 1 ,40848   ,357,357,357
BEGIN DESCRIPTION:
North Deep Creek 107.0
END DESCRIPTION:
XS GIS Cut Line= 4
      1515326.39       874789.24       1515334.1       874588.82
      1515276.29       874361.44      1515191.51       874226.55
#Sta/Elev= 30
  4846.8  847.54    4875  843.73  4906.1  837.69  4926.1  833.18  4946.6  827.23
  4957.2  823.47  4970.8  819.98  4982.6  816.22  4983.4  805.56  4984.5  802.56
  5015.5  802.56  5016.6  805.56  5029.2  806.32  5036.5  809.46  5041.9  811.18
  5052.9  812.66  5061.3  812.04    5095  811.65  5150.5  812.96    5180  812.33
  5275.1  812.14  5294.3  813.33  5317.7  816.52  5333.9  822.16  5351.7  827.73
  5388.5  837.59  5396.2  839.75  5399.7  841.13  5413.1  843.16  5441.3  848.42
#Mann= 3 ,-1 , 0
  4846.8     .14       0  4983.4    .045       0  5016.6     .14       0
Bank Sta=4983.4,5016.6
Exp/Cntr=0.3,0.1

Type RM Length L Ch R = 1 ,40491   ,676,676,676
BEGIN DESCRIPTION:
North Deep Creek 106.0
END DESCRIPTION:
XS GIS Cut Line= 4
       1516062.5       874789.24      1515923.74       874677.46
      1515337.96       874330.61      1515222.34       874222.71
#Sta/Elev= 30
  4499.2  838.13  4563.8  830.56  4589.9  826.61  4609.3  822.66  4623.4   820.6
  4646.2  813.92    4668   811.7  4702.5   810.9  4869.9  810.63    4953  811.66
  4958.1  811.38  4976.3  805.36  4977.8  802.36  5022.2  802.36  5023.7  805.36
  5027.9  811.62  5048.2  809.98  5096.4  808.92  5114.6  811.05  5176.2  809.98
  5298.3  811.81    5353  811.48  5384.5  812.68    5397  811.55    5409  811.74
  5419.7  814.42  5436.9   820.8  5456.4  826.12  5469.7  830.63  5516.3  840.76
#Mann= 3 ,-1 , 0
  4499.2     .07       0  4976.3    .045       0  5023.7     .14       0
#XS Ineff= 2 , 0
       0  4846.4  825.92               0
Permanent Ineff=
       F       F
Bank Sta=4976.3,5023.7
Exp/Cntr=0.3,0.1

Type RM Length L Ch R = 1 ,39815   ,624,624,624
BEGIN DESCRIPTION:
North Deep Creek 105.0
END DESCRIPTION:
XS GIS Cut Line= 4
      1516413.17       874188.02      1516197.36        874114.8
      1515596.16       873737.12      1515461.25       873609.92
#Sta/Elev= 30
  4433.7  835.45  4498.2  827.65    4553  823.74  4579.8  822.69  4618.7  818.56
  4631.8  816.34  4657.3  816.52  4661.6  815.47  4723.7  810.88  4798.7  808.95
  4902.7  810.27  4934.6   809.9  4949.6  810.66  4963.5  809.29  4976.3  805.16
  4977.8  802.16  5022.2  802.16  5023.7  805.16  5036.2  810.29  5038.9  810.46
  5139.9  808.16    5234  808.34  5282.1  809.69  5353.6   809.4  5380.1  810.08
  5393.9  815.48  5413.8  827.89  5432.5   838.4  5457.7  846.08    5557  859.98
#Mann= 4 ,-1 , 0
  4433.7     .07       0  4963.5     .14       0  4976.3    .045       0
  5023.7     .14       0
Bank Sta=4976.3,5023.7
Exp/Cntr=0.3,0.1

Type RM Length L Ch R = 1 ,39191   ,364,364,364
BEGIN DESCRIPTION:
North Deep Creek 104.0
END DESCRIPTION:
XS GIS Cut Line= 4
      1516767.75       873706.29      1516613.57       873679.31
      1516131.85       873351.74       1516085.6       873293.93
#Sta/Elev= 30
  4344.2  847.64  4356.9  845.14  4382.6  841.69  4405.3  835.94  4426.4  826.25
  4436.4  822.46  4468.5  813.34  4484.1  810.85  4505.6  808.79  4524.3  807.85
  4554.7  807.28  4638.7  808.45  4677.8     808  4813.7  808.07  4893.1  808.93
  4937.5  808.87  4958.3  809.38  4971.9  807.72  4976.3  804.64  4977.8  801.64
  5022.2  801.64  5023.7  804.64  5057.7  807.82  5081.5  807.19  5094.8  807.68
    5099  809.04  5114.2  821.01  5133.4  831.81    5141  837.39  5157.3  844.73
#Mann= 4 ,-1 , 0
  4344.2     .07       0  4893.1     .14       0  4976.3    .045       0
  5023.7     .14       0
#XS Ineff= 2 , 0
       0  4667.1  828.41               0
Permanent Ineff=
       F       F
Bank Sta=4976.3,5023.7
Exp/Cntr=0.3,0.1

Type RM Length L Ch R = 1 ,38827   ,275,275,275
BEGIN DESCRIPTION:
North Deep Creek 103.0
END DESCRIPTION:
XS GIS Cut Line= 3
      1516640.52       873355.56      1516447.86       873170.61
       1516436.3       873074.27
#Sta/Elev= 30
  4707.5  827.78  4720.9  825.61  4725.4  825.64  4740.7     822  4745.7  821.87
  4759.5  817.93  4784.3  810.11  4799.4  806.81  4819.4  805.86  4824.2  804.88
    4840  807.08  4863.7  807.38  4879.1  806.57  4899.4  806.96  4905.8   807.6
  4926.1   807.8  4942.1  807.44  4968.3  808.46  4976.6  807.76  4978.7  803.51
    4980  800.51    5020  800.51  5021.3  803.51    5023  809.83  5030.6  811.39
  5032.3   812.1    5046  821.84  5049.9  824.98    5057  829.07  5071.6  840.86
#Mann= 4 ,-1 , 0
  4707.5     .07       0  4819.4     .14       0  4978.7    .045       0
  5021.3     .14       0
Bank Sta=4978.7,5021.3
Exp/Cntr=0.3,0.1

Type RM Length L Ch R = 1 ,38552   ,545,545,545
BEGIN DESCRIPTION:
North Deep Creek 102.0
END DESCRIPTION:
XS GIS Cut Line= 4
      1516786.98       873359.41      1516725.34       873232.27
      1516702.21        873112.8      1516632.87       873008.78
#Sta/Elev= 30
  4760.2  833.84  4767.5   833.4  4783.4  831.45  4788.5   831.2  4825.7   826.5
    4845  823.24  4869.4  817.56  4882.8   814.9  4892.7  812.42  4918.5  807.55
  4942.8  806.81  4954.6  807.56    4957   806.9  4967.4  805.78  4980.2  803.86
    4981  802.95  4982.2  799.95  5017.8  799.95    5019  802.95  5023.2  807.13
  5030.2   808.7  5051.6  808.25  5067.1  816.52  5070.5  817.98  5080.4  824.62
  5090.6  828.17  5093.8  829.78  5113.7  837.34  5131.5  843.44  5148.2  848.44
#Mann= 4 ,-1 , 0
  4760.2     .07       0  4942.8     .14       0    4981    .045       0
    5019     .14       0
Bank Sta=4981,5019
Exp/Cntr=0.3,0.1

Type RM Length L Ch R = 1 ,38007   ,432,432,432
BEGIN DESCRIPTION:
North Deep Creek 101.0
END DESCRIPTION:
XS GIS Cut Line= 4
      1517141.56       873386.39      1517222.48       873159.05
      1517222.48       872987.55      1517264.86       872877.76
#Sta/Elev= 30
    4636  840.01  4665.1  838.48  4701.3   835.6  4729.6  832.58    4752  829.35
  4771.3  827.43  4798.5  822.21  4811.1   819.4    4822  817.49  4845.6  811.61
  4863.3  807.94  4891.6  806.68  4901.1  807.03    4923   806.8  4938.3  807.33
    4961  807.87  4972.5  807.78  4976.3  802.73  4977.8  799.73  5022.2  799.73
  5023.7  802.73  5043.2  807.97  5049.5  808.12  5061.7  812.68  5067.2  814.36
  5069.2  815.83    5085  821.89  5099.4  825.19  5131.9  831.43  5166.5  833.86
#Mann= 4 ,-1 , 0
    4636     .07       0  4938.3     .14       0  4976.3    .045       0
  5023.7     .14       0
Bank Sta=4976.3,5023.7
Exp/Cntr=0.5,0.3

Type RM Length L Ch R = 1 ,37575   ,123,123,123
BEGIN DESCRIPTION:
Myers Rd (NDC) us
END DESCRIPTION:
XS GIS Cut Line= 4
      1517453.62       873718.65      1517568.91       873372.78
      1517639.57       873108.76      1517632.13       872867.06
#Sta/Elev= 30
  4312.7  853.87  4317.1  853.08  4362.4   850.5  4384.6  848.37  4407.5  845.63
  4421.9  843.33  4436.2  840.12  4459.7  838.52  4470.1  836.28  4482.8  832.59
  4600.8   821.7  4638.3  814.27  4664.7  809.76    4695  808.01  4727.5  807.47
  4900.8  806.31  4930.5  806.83  4967.2  807.95    4980   807.2    4984   798.7
    5016   798.7    5020   807.2  5022.5  807.56    5035  814.01    5064  821.94
    5124  832.61  5153.8  836.23  5164.8  838.17  5177.7  839.25  5192.4  841.34
#Mann= 4 ,-1 , 0
  4312.7     .07       0  4930.5     .14       0    4980    .045       0
    5020     .14       0
#XS Ineff= 2 , 0
       0  4939.5  808.61  5060.5       0  816.59
Permanent Ineff=
       F       F
Bank Sta=4980,5020
Exp/Cntr=0.5,0.3

Type RM Length L Ch R = 3 ,37525   ,,,
BEGIN DESCRIPTION:
Myers Rd (NDC) tor
Structure ID: LDS_NDC_09
Approximate Survey Structure
END DESCRIPTION:
Bridge Culvert--1,0,-1,-1, 0
Deck Dist Width WeirC Skew NumUp NumDn MinLoCord MaxHiCord MaxSubmerge Is_Ogee
40.5,19,3,0, 16, 16, , , 0.95, 0, 1,1,,
  4337.3  4466.5  4617.2  4694.9    4730  4778.4  4873.6  4919.8    4980    4980
    5020    5020  5062.1  5095.7  5271.6    5331
  841.77  829.48  816.74  812.22  810.78  809.56  808.87  809.38   812.5   812.5
  814.58  814.58  816.76  819.65  838.99  843.94
   778.7   778.7   778.7   778.7   778.7   778.7   778.7   778.7   778.7   809.9
  811.86   778.7   778.7   778.7   778.7   778.7
  4337.3  4466.5  4617.2  4694.9    4730  4778.4  4873.6  4919.8    4980    4980
    5020    5020  5062.1  5095.7  5271.6    5331
  841.77  829.48  816.74  812.22  810.78  809.56  808.87  809.38   812.5   812.5
  814.58  814.58  816.76  819.65  838.99  843.94
   778.7   778.7   778.7   778.7   778.7   778.7   778.7   778.7   778.7   809.9
  811.86   778.7   778.7   778.7   778.7   778.7
BR Coef= 1 , 1 , 0 ,1.25, 0 ,,,0.8,-1,2,0,
WSPro=,,,, 1 ,,,, 0 ,,,, 0 ,,,,-1 ,-1 ,-1 , 0 , 0 , 0 , 0 , 0
BC Design=,, 0 ,, 0 ,,,,,,
BC HTab HWMax=853.87

Type RM Length L Ch R = 1 ,37452   ,230,230,230
BEGIN DESCRIPTION:
Myers Rd (NDC) ds
END DESCRIPTION:
XS GIS Cut Line= 5
      1517639.56       873714.93      1517702.78       873439.71
      1517732.53       873153.38      1517758.56       873038.11
      1517758.56       872796.44
#Sta/Elev= 30
  4365.9  841.28    4446   832.6  4491.4  830.16  4528.6  825.18    4573  822.24
    4578  819.83  4590.8  821.45  4624.4  819.78  4638.7  815.43  4649.6  809.58
  4656.1  807.83  4686.6  806.92  4706.8   809.3  4734.4  809.56    4771  806.96
  4791.6  807.81  4816.4  806.42  4928.1  806.44  4968.6  808.76    4980  806.95
    4984  798.45    5016  798.45    5020  800.98  5040.1  802.52  5068.6  812.82
  5086.2  815.27    5108  815.57  5158.7  820.27  5280.4  834.41    5296  835.79
#Mann= 4 ,-1 , 0
  4365.9     .14       0    4980    .045       0    5020     .14       0
  5280.4     .14       0
#XS Ineff= 2 , 0
       0  4916.5  809.28  5083.5       0   818.7
Permanent Ineff=
       F       F
Bank Sta=4980,5020
Exp/Cntr=0.5,0.3

Type RM Length L Ch R = 1 ,37222   ,358,358,358
BEGIN DESCRIPTION:
North Deep Creek 100.0
END DESCRIPTION:
XS GIS Cut Line= 6
      1518212.24       873562.44      1518059.76       873409.96
       1517966.8        873097.6      1517903.59       872844.74
      1517799.47       872770.37        1517766.       872725.75
#Sta/Elev= 30
  4466.1  847.85  4572.4   832.4  4616.4  823.14  4629.8  819.85  4674.2  811.79
  4692.9  809.23  4750.9  806.94  4805.2  806.76  4822.7  805.92  4832.8  806.68
  4859.7  806.12  4890.9  807.48  4930.8  806.64  4950.9  808.54  4956.4  807.26
  4957.6     808  4963.5  807.32  4975.8  800.59  4977.3  797.59  5022.7  797.59
  5024.2  800.59  5028.6  805.89  5040.7  807.65  5072.5  809.53  5115.9  813.64
  5123.3   813.4  5176.2  818.54  5276.1  823.43  5322.8   827.2    5452   842.9
#Mann= 4 ,-1 , 0
  4466.1      .1       0  4616.4     .14       0  4975.8    .045       0
  5024.2     .14       0
Bank Sta=4975.8,5024.2
Exp/Cntr=0.3,0.1

Type RM Length L Ch R = 1 ,36864   ,442,442,442
BEGIN DESCRIPTION:
North Deep Creek 99.0
END DESCRIPTION:
XS GIS Cut Line= 4
       1518405.6        873231.5      1518271.72       872930.27
      1518108.11       872829.87      1517818.03       872740.61
#Sta/Elev= 30
  4738.8  827.05  4754.8  823.75  4776.3  821.25  4802.5  811.35  4807.3   810.3
  4814.8  808.67  4818.9  806.81  4823.5   806.7  4838.5   804.3  4845.5  804.81
  4858.1  804.49  4866.8  805.35  4958.6  805.87  4963.3  805.13  4975.8  799.89
  4977.3  796.89  5022.7  796.89  5024.2  799.89  5032.6     805  5052.4  807.28
  5097.6  807.87  5143.8  806.95  5208.9  809.27  5259.2  813.87  5383.6   822.4
  5448.2  828.32  5456.4  829.82  5467.3  830.04  5483.3  831.84  5563.9  837.54
#Mann= 4 ,-1 , 0
  4738.8      .1       0  4807.3     .14       0  4975.8    .045       0
  5024.2     .14       0
Bank Sta=4975.8,5024.2
Exp/Cntr=0.3,0.1

Type RM Length L Ch R = 1 ,36422   ,309,309,309
BEGIN DESCRIPTION:
North Deep Creek 98.0
END DESCRIPTION:
XS GIS Cut Line= 5
      1518721.66       873093.86      1518636.14        872956.3
      1518468.81       872833.59      1518122.98       872766.65
      1517836.69       872710.88
#Sta/Elev= 30
  4879.7  833.15  4899.3  827.21  4926.2  820.37  4957.9  808.83  4958.4  808.06
  4974.2  805.66  4975.8  799.63  4977.3  796.63  5022.7  796.63  5024.2  799.63
  5029.3  806.42  5045.5  807.18  5069.4  806.46  5101.5   806.5  5142.6  805.34
  5172.1   806.7  5178.1  806.17    5199  806.85  5203.8   806.2  5227.2  806.04
  5288.7   806.5  5389.6  805.86  5484.1  806.98  5530.2  808.79  5593.5   812.2
  5715.7  825.72    5752  828.55  5786.3  832.63  5844.5  835.63  5893.1   839.2
#Mann= 4 ,-1 , 0
  4879.7      .1       0  4975.8    .045       0  5024.2      .1       0
  5069.4     .14       0
#XS Ineff= 2 , 0
       0                  5429.1       0  822.88
Permanent Ineff=
       F       F
Bank Sta=4975.8,5024.2
Exp/Cntr=0.3,0.1

Type RM Length L Ch R = 1 ,36113   ,337,337,337
BEGIN DESCRIPTION:
North Deep Creek 97.0
END DESCRIPTION:
XS GIS Cut Line= 4
       1519067.5       872803.84      1518796.04       872759.21
      1518163.88       872733.18       1517866.4       872688.56
#Sta/Elev= 30
  4797.8  844.66  4820.7  841.41  4850.5  834.32  4894.7  812.08  4907.3   809.5
  4924.9     808    4962  806.54  4975.8  799.48  4977.3  796.48  5022.7  796.48
  5024.2  799.48  5029.1  804.16  5042.6  805.27  5077.5  801.57  5103.5  801.15
  5114.9  803.81  5166.8  804.94  5255.7  804.72  5289.7  805.88  5377.2   806.1
  5411.3   805.4  5455.6  806.42  5497.8  804.88  5507.2  805.83  5656.9  807.53
  5745.4  812.15  5857.7   827.4  5958.2  836.68  5971.3  836.37  6006.4  839.14
#Mann= 4 ,-1 , 0
  4797.8      .1       0  4975.8    .045       0  5024.2      .1       0
  5077.5     .14       0
#XS Ineff= 2 , 0
       0                  5377.6       0  825.37
Permanent Ineff=
       F       F
Bank Sta=4975.8,5024.2
Exp/Cntr=0.5,0.3

Type RM Length L Ch R = 1 ,35776   ,161,161,161
BEGIN DESCRIPTION:
Old US 421 (NDC) us
END DESCRIPTION:
XS GIS Cut Line= 6
      1519061.96       872513.79      1518911.32       872500.77
      1518760.71       872474.74      1518520.87       872513.79
      1518121.12       872569.57      1517901.71       872565.85
#Sta/Elev= 30
  4734.6  844.19    4762  840.48    4791  837.48  4838.1  827.36  4906.8  806.25
  4925.5  804.54    4981     804    4985   796.1    5015   796.1    5019     804
  5076.8  803.06  5176.3  803.46  5216.3  804.57  5224.3  806.03  5240.7  806.47
  5273.3   805.4  5325.3  807.86  5379.4  806.77  5459.2  810.01  5484.5  808.54
  5523.4  810.99  5540.5  810.19  5607.7  811.45  5678.9   814.7  5716.2  817.54
  5775.5  825.92  5837.7  836.72  5845.3  836.08  5896.9  841.21  5904.7  841.89
#Mann= 5 ,-1 , 0
  4734.6      .1       0    4762     .14       0    4981    .045       0
    5019     .14       0  5896.9     .14       0
#XS Ineff= 2 , 0
       0    4828   816.1    5172       0  816.66
Permanent Ineff=
       F       F
Bank Sta=4981,5019
Exp/Cntr=0.5,0.3

Type RM Length L Ch R = 3 ,35689   ,,,
BEGIN DESCRIPTION:
Old US 421 (NDC) tor
Structure ID: LDS_NDC_08
Approximate Survey Structure
END DESCRIPTION:
Bridge Culvert--1,0,-1,-1, 0
Deck Dist Width WeirC Skew NumUp NumDn MinLoCord MaxHiCord MaxSubmerge Is_Ogee
71,32,3,0, 14, 14, , , 0.95, 0, 1,1,,
  4584.7    4899    4899    5101    5101  5151.6  5204.8  5347.6  5423.7  5526.3
  5598.4  5693.9  5820.9  5910.3
   816.1   816.1   816.1   816.1   816.1   816.1  816.57  818.85  820.89  823.64
  826.42  830.97  838.19  843.85
   776.1   776.1   811.6   811.6   776.1   776.1   776.1   776.1   776.1   776.1
   776.1   776.1   776.1   776.1
  4584.7    4899    4899    5101    5101  5151.6  5204.8  5347.6  5423.7  5526.3
  5598.4  5693.9  5820.9  5910.3
   816.1   816.1   816.1   816.1   816.1   816.1  816.57  818.85  820.89  823.64
  826.42  830.97  838.19  843.85
   776.1   776.1   811.6   811.6   776.1   776.1   776.1   776.1   776.1   776.1
   776.1   776.1   776.1   776.1
Pier Skew, UpSta & Num, DnSta & Num=  ,4949.5, 2 ,4949.5, 2 , 0 , 0 , 0 ,0,0
       3       3
  804.14   811.6
       3       3
  810.38   811.6
Pier Skew, UpSta & Num, DnSta & Num=  ,5050.5, 2 ,5050.5, 2 , 0 , 0 , 0 ,0,0
       3       3
   803.3   811.6
       3       3
  805.11   811.6
Abutment Skew #Up #Dn= , 2 , 2
    4899  4908.3
   811.6  806.05
    4899  4908.3
   811.6  814.56
Abutment Skew #Up #Dn= , 2 , 2
  5091.8    5101
  803.46   811.6
  5091.8    5101
  804.46   811.6
BR Coef= 1 , 1 , 0 ,1.25, 0 ,,,0.8,0,2,0,
WSPro=,,,, 1 ,,,, 0 ,,,, 0 ,,,,-1 ,-1 ,-1 , 0 , 0 , 0 , 0 , 0
BC Design=,, 0 ,, 0 ,,,,,,
BC HTab HWMax=844.19

Type RM Length L Ch R = 1 ,35615   ,206,206,206
BEGIN DESCRIPTION:
Old US 421 (NDC) ds
END DESCRIPTION:
XS GIS Cut Line= 6
      1519147.42       872266.51      1518799.76       872327.86
      1518543.18       872365.05      1518470.67       872363.19
      1518359.11       872327.86      1518292.17       872244.19
#Sta/Elev= 30
    4578   823.3  4599.5  822.55  4617.8  819.44  4641.7   818.9  4666.8  816.92
  4704.9   815.6  4783.8  815.08  4842.6  815.65  4915.5  814.54    4945  811.78
    4958  807.47  4975.1  803.01    4981  803.75    4985  795.85    5015  795.85
    5019  803.75  5020.6  804.54  5029.1  805.43  5091.1  804.45  5113.2  804.82
  5156.1  809.06  5170.1   809.5  5232.9  816.06  5270.7  815.98  5337.6  818.97
  5403.1  825.11  5415.2  828.69  5439.9  833.03  5454.8  834.74    5487  836.44
#Mann= 3 ,-1 , 0
    4578     .09       0    4981    .045       0    5019     .09       0
#XS Ineff= 2 , 0
       0    4841   816.1    5159       0  816.21
Permanent Ineff=
       F       F
Bank Sta=4981,5019
Exp/Cntr=0.5,0.3
