HEC-RAS study North Deep Creek.prj: North Deep Creek Limited Detail Study

--- North Deep Creek.g01 (geometry) --- (continued)

Type RM Length L Ch R = 1 ,35409   ,186,186,186
BEGIN DESCRIPTION:
North Deep Creek 95.0
END DESCRIPTION:
XS GIS Cut Line= 4
       1519041.5       872249.78      1518781.17       872160.53
       1518647.3       872086.15      1518580.37        871993.2
#Sta/Elev= 30
  4678.2  817.05  4729.2  816.24  4748.2  814.98  4769.6  812.33  4794.2   810.8
  4836.4  807.17  4886.4  804.19  4911.8  803.33    4939  803.11    4966  799.04
  4980.3  798.12  4980.6  797.43  4981.8  794.43  5018.2  794.43  5019.4  797.43
    5025  804.34  5032.8  804.69  5058.1  804.39  5095.9  801.67  5121.9  802.41
  5140.1  804.69  5144.4  806.65  5150.2  810.75  5166.5  820.32  5175.8  821.57
  5180.3   825.1  5198.1  837.71  5209.7  843.91  5212.4  844.84  5221.1   846.3
#Mann= 4 ,-1 , 0
  4678.2     .09       0  4769.6    .115       0  4980.6    .045       0
  5019.4    .115       0
Bank Sta=4980.6,5019.4
Exp/Cntr=0.3,0.1

Type RM Length L Ch R = 1 ,35223   ,298,298,298
BEGIN DESCRIPTION:
North Deep Creek 94.0
END DESCRIPTION:
XS GIS Cut Line= 3
      1519071.21       872223.74      1518803.48       871989.47
      1518729.11       871885.36
#Sta/Elev= 30
  4619.6  818.58  4637.7  818.82  4650.5  818.52  4657.8  817.85  4669.6   817.3
  4684.3  816.19  4704.2  814.96    4709  814.87  4714.6  814.82  4732.9  813.66
    4758  810.24  4786.3  807.79  4807.9  805.63    4815  805.44    4822  804.83
  4863.5  803.17  4887.6  802.97  4920.6  804.21  4926.9  803.77    4958  800.19
  4975.4  798.53  4978.2  797.27  4979.6  794.27  5020.4  794.27  5021.8  797.27
  5041.4  818.19  5049.9  822.45  5067.3  829.72  5077.6  829.47  5103.3  831.55
#Mann= 4 ,-1 , 0
  4619.6     .09       0    4709    .115       0  4978.2    .045       0
  5021.8    .115       0
Bank Sta=4978.2,5021.8
Exp/Cntr=0.3,0.1

Type RM Length L Ch R = 1 ,34925   ,525,525,525
BEGIN DESCRIPTION:
North Deep Creek 93.0
END DESCRIPTION:
XS GIS Cut Line= 4
       1519108.4       872205.11      1519100.96       871996.91
       1519048.9       871825.86      1519041.46       871651.05
#Sta/Elev= 30
  4638.2  819.64  4649.2  818.87  4708.5  815.17  4722.9  813.94  4735.8  813.66
  4761.2   811.5  4790.3  809.53  4836.4  804.78  4860.7  803.21  4873.4  802.62
  4909.4  803.69  4969.3  802.54  4978.2  796.85  4979.6  793.85  5020.4  793.85
  5021.8  796.85  5021.9  799.22  5041.7  803.91  5050.4  804.66  5060.8  807.35
  5067.5  812.48    5085  824.39    5090  830.41  5117.3  849.97  5132.7  857.39
  5143.8  860.65  5156.4  863.84  5171.4  866.97  5189.4  871.24  5200.3  873.01
#Mann= 4 ,-1 , 0
  4638.2     .09       0  4649.2    .115       0  4978.2    .045       0
  5021.8    .115       0
Bank Sta=4978.2,5021.8
Exp/Cntr=0.3,0.1

Type RM Length L Ch R = 1 ,34400   ,436,436,436
BEGIN DESCRIPTION:
North Deep Creek 92.0
END DESCRIPTION:
XS GIS Cut Line= 4
      1519662.85       871911.57       1519597.4       871806.12
      1519546.49       871686.12       1519459.2       871584.28
#Sta/Elev= 30
  4775.9  828.16  4792.2  825.59  4804.7   823.9    4832  819.28  4842.5  817.96
  4847.7  817.01  4853.9  815.64  4876.5  811.35  4896.8  807.73  4910.9  806.89
  4932.1  804.98  4943.4  802.12  4945.8  801.82  4948.7  802.04  4956.7  803.13
  4968.9  802.81  4972.7  802.14  4980.6  796.18  4981.8  793.18  5018.2  793.18
  5019.4  796.18  5025.2  805.55  5049.3  808.29  5049.9  808.49  5069.4  821.49
  5089.3  827.66  5128.7  846.31  5131.6  847.32  5145.6   849.3  5164.5  853.04
#Mann= 4 ,-1 , 0
  4775.9      .1       0  4876.5    .115       0  4980.6    .045       0
  5019.4    .115       0
Bank Sta=4980.6,5019.4
Exp/Cntr=0.3,0.1

Type RM Length L Ch R = 1 ,33964   ,265,265,265
BEGIN DESCRIPTION:
North Deep Creek 91.0
END DESCRIPTION:
XS GIS Cut Line= 4
      1520084.69        871911.6      1519990.13       871697.03
      1519950.13       871355.21      1519888.32       871206.15
#Sta/Elev= 30
  4678.8  837.84  4711.6  834.91  4717.1  833.56  4745.1  829.33  4763.3  825.86
  4778.6  823.87  4794.1  819.91  4820.5  815.35    4843  812.26  4855.6  809.74
  4882.9  806.36  4901.5  804.76  4927.8  803.46  4971.8  802.23  4975.8  796.02
  4977.3  793.02  5022.7  793.02  5024.2  796.02  5028.1   805.6    5040  804.22
  5115.6  804.28  5257.4  810.91  5277.4  821.23  5302.2  834.98  5312.6  839.29
  5324.3  843.41  5335.7  846.27  5347.2  849.87  5391.1  859.68  5418.8  860.68
#Mann= 3 ,-1 , 0
  4678.8      .1       0  4975.8    .045       0  5024.2    .115       0
Bank Sta=4975.8,5024.2
Exp/Cntr=0.3,0.1

Type RM Length L Ch R = 1 ,33699   ,482,482,482
BEGIN DESCRIPTION:
North Deep Creek 90.0
END DESCRIPTION:
XS GIS Cut Line= 4
      1520397.37       871744.27      1520248.31       871591.58
      1520161.04       871431.57      1519971.97       871184.33
#Sta/Elev= 30
  4641.1  835.15  4654.2  833.93  4665.8  834.74  4715.1   827.9  4724.4  827.79
  4762.7  823.43  4785.6  820.15  4864.3  805.31  4895.8  802.84  4911.4  803.31
  4933.8  801.92  4944.4  797.58  4955.2  800.46  4976.9  799.24  4980.4  795.93
  4981.6  792.93  5018.4  792.93  5019.6  795.93  5031.2   803.7  5082.8  804.63
  5130.3  802.99  5172.4  803.65  5194.9  806.63  5217.4  813.48  5227.4  818.02
  5238.6  820.89  5258.6   829.9  5291.4  841.88  5319.2   849.8    5348  855.46
#Mann= 4 ,-1 , 0
  4641.1      .1       0  4980.4    .045       0  5019.6      .1       0
  5172.4    .115       0
Bank Sta=4980.4,5019.6
Exp/Cntr=0.3,0.1

Type RM Length L Ch R = 1 ,33217   ,428,428,428
BEGIN DESCRIPTION:
North Deep Creek 89.0
END DESCRIPTION:
XS GIS Cut Line= 4
      1520713.77        871609.8      1520717.41       871442.48
      1520535.59       871147.94      1520390.13       870933.39
#Sta/Elev= 30
  4567.3  846.38  4605.5  838.85  4649.2  828.26  4721.8  805.02  4736.9  801.53
  4823.7  802.27  4914.1  801.77  4959.3   803.3  4975.5  795.37    4977  792.37
    5023  792.37  5024.5  795.37    5028  802.76  5048.9  802.41  5059.5  801.04
  5112.8   801.6  5135.3  800.11  5155.4  800.72  5170.4  804.01  5176.2  804.83
  5186.5  808.71  5200.5  812.03  5219.1  821.75    5227  828.25  5250.7  843.33
  5262.1   849.2  5282.3  857.72  5295.5  861.58  5307.1  866.13    5340  873.55
#Mann= 5 ,-1 , 0
  4567.3      .1       0  4914.1     .13       0  4975.5    .045       0
  5024.5     .13       0  5170.4     .13       0
Bank Sta=4975.5,5024.5
Exp/Cntr=0.3,0.1

Type RM Length L Ch R = 1 ,32789   ,327,327,327
BEGIN DESCRIPTION:
North Deep Creek 88.0
END DESCRIPTION:
XS GIS Cut Line= 4
      1521226.49       871435.19      1521131.95       871329.76
      1520873.77       870893.39      1520826.49       870733.36
#Sta/Elev= 30
    4417   839.3  4465.6  834.59    4494   830.4  4525.5  828.08  4598.7  802.73
  4610.3  801.15  4659.5  799.92  4683.2  801.81  4716.9  801.84  4728.9  800.83
    4850  802.46  4914.5  800.69  4949.8  801.55  4970.1  799.97  4975.5  794.95
    4977  791.95    5023  791.95  5024.5  794.95  5026.2  801.19  5067.4  801.41
    5078  803.86  5100.5  805.41  5117.4  809.44  5136.5  815.52  5147.7  820.56
    5176  836.49  5184.4  842.92  5189.2  847.78  5216.8  866.43  5232.5   872.4
#Mann= 4 ,-1 , 0
    4417      .1       0  4716.9     .13       0  4975.5    .045       0
  5024.5     .13       0
Bank Sta=4975.5,5024.5
Exp/Cntr=0.3,0.1

Type RM Length L Ch R = 1 ,32462   ,591,591,591
BEGIN DESCRIPTION:
North Deep Creek 87.0
END DESCRIPTION:
XS GIS Cut Line= 4
      1521444.65       871278.81      1521335.59       871151.57
      1521161.05       870755.21      1521110.12       870646.08
#Sta/Elev= 30
  4392.7  839.98  4419.5  837.37    4472  827.99  4491.4  826.37  4505.2  820.64
  4540.4  809.57  4560.4  802.24  4606.1  800.42  4662.1  800.26  4703.5  800.66
  4758.3  799.67  4849.5  800.94  4884.7  800.05  4927.8  800.35  4944.1  801.63
    4956  803.75  4970.2   802.8  4973.6  801.65  4980.4  794.81  4981.6  791.81
  5018.4  791.81  5019.6  794.81  5021.8  800.36  5032.3  804.61  5044.4  813.78
  5058.6  822.67  5067.3  830.71    5093  847.97  5103.1  853.01  5113.8  856.79
#Mann= 4 ,-1 , 0
  4392.7      .1       0  4662.1     .13       0  4980.4    .045       0
  5019.6     .13       0
Bank Sta=4980.4,5019.6
Exp/Cntr=0.3,0.1

Type RM Length L Ch R = 1 ,31871   ,440,440,440
BEGIN DESCRIPTION:
North Deep Creek 86.0
END DESCRIPTION:
XS GIS Cut Line= 4
      1521819.23       870995.23      1521808.32       870773.39
      1521677.41       870497.02      1521648.32       870355.19
#Sta/Elev= 30
    4436  838.05  4447.8  837.56  4459.7  836.16    4512  829.07  4543.4  823.47
  4554.9  820.93  4582.9  816.74  4612.9  813.94  4647.3  808.89  4671.1   805.9
  4684.8  804.41  4707.9  802.66    4774  800.14  4805.9  800.22  4846.7  798.76
  4894.5  798.44    4932  798.66  4952.6  799.76  4970.6   801.4  4975.5  793.89
    4977  790.89    5023  790.89  5024.5  793.89  5024.8  800.14  5034.5  801.41
  5043.3  803.61  5082.8  831.17    5086  832.83  5087.9  834.24  5108.7  840.49
#Mann= 5 ,-1 , 0
    4436      .1       0  4554.9     .07       0  4894.5     .13       0
  4975.5    .045       0  5024.5     .13       0
Bank Sta=4975.5,5024.5
Exp/Cntr=0.3,0.1

Type RM Length L Ch R = 1 ,31431   ,578,578,578
BEGIN DESCRIPTION:
North Deep Creek 85.0
END DESCRIPTION:
XS GIS Cut Line= 4
      1522273.78       870686.11      1522146.51       870555.21
      1522077.41       870293.39      1522019.26       870206.15
#Sta/Elev= 30
  4596.1  821.66  4634.8  819.54  4654.9  817.24  4667.6  816.22  4674.5  815.09
  4750.7  807.41  4757.5  806.12  4778.9  803.89  4795.2  801.77    4830  799.84
  4884.2  799.29  4918.1   797.5  4945.4  795.77  4959.5  796.91  4972.5  798.91
  4975.3  796.41  4975.5  792.96    4977  789.96    5023  789.96  5024.5  792.96
  5037.6  799.09    5043  799.95    5063  800.35  5076.3  804.59  5083.5  807.08
  5097.9  813.44  5116.5     823  5121.4  825.12  5138.3  831.96  5154.3  836.87
#Mann= 4 ,-1 , 0
  4596.1     .07       0  4918.1     .13       0  4975.5    .045       0
  5024.5     .13       0
Bank Sta=4975.5,5024.5
Exp/Cntr=0.3,0.1

Type RM Length L Ch R = 1 ,30853   ,452,452,452
BEGIN DESCRIPTION:
North Deep Creek 84.0
END DESCRIPTION:
XS GIS Cut Line= 4
      1522699.23       870555.18      1522622.87       870191.57
      1522477.42       869900.66      1522462.87        869602.5
#Sta/Elev= 30
    4367  816.83  4403.8  814.38  4557.4  806.85  4620.6  804.97    4639  803.86
  4692.9  801.91  4729.8  801.33  4756.5  800.04  4777.8   799.9  4819.2  797.94
  4880.8  797.12  4893.9  796.71    4917  797.73  4932.5  795.31  4940.6  794.49
  4954.5  794.55  4971.5  792.86  4975.5  792.85    4977  789.85    5023  789.85
  5024.5  792.85  5025.5  794.06  5032.5   797.7  5055.4  798.04  5090.5  799.71
  5156.6   805.1  5218.6  812.29  5290.3  823.17  5350.9  830.43  5362.3  831.41
#Mann= 4 ,-1 , 0
    4367     .07       0  4880.8     .13       0  4975.5    .045       0
  5024.5     .07       0
Bank Sta=4975.5,5024.5
Exp/Cntr=0.3,0.1

Type RM Length L Ch R = 1 ,30401   ,377,377,377
BEGIN DESCRIPTION:
North Deep Creek 83.0
END DESCRIPTION:
XS GIS Cut Line= 4
      1523142.86        870206.1      1522942.87       870053.39
      1522917.42       869827.93      1522891.96       869682.46
#Sta/Elev= 30
  4593.5  816.01  4655.8   812.3  4666.2  810.92  4703.8  808.11  4738.6  807.13
  4782.5  806.89  4797.5   804.7  4835.7  801.89    4839  801.94  4868.7  798.09
  4882.3  797.21  4890.7  797.09  4931.6  796.19  4947.8  797.29  4973.1  792.78
  4974.7  789.78  5025.3  789.78    5027  792.78  5027.6  794.75  5035.2  798.11
  5050.6  797.46  5073.8  800.53  5094.8  806.58  5105.7  810.58  5114.5  814.28
  5120.1  817.44  5138.6  825.89    5155  829.01  5203.5   837.8  5219.7  838.92
#Mann= 5 ,-1 , 0
  4593.5      .1       0  4890.7     .13       0  4973.1    .045       0
    5027     .13       0    5155     .07       0
Bank Sta=4973.1,5027
Exp/Cntr=0.3,0.1

Type RM Length L Ch R = 1 ,30024   ,254,254,254
BEGIN DESCRIPTION:
North Deep Creek 82.0
END DESCRIPTION:
XS GIS Cut Line= 4
      1523386.52       870137.05      1523342.88       869933.38
      1523259.24       869798.84      1523219.24       869667.92
#Sta/Elev= 30
    4690  819.46  4730.9  815.63  4750.7  814.51  4764.4  813.18  4798.6  811.36
  4834.2  810.43  4848.4  810.48  4892.2  808.29  4925.7  803.87  4938.8  801.85
  4959.7  799.38    4969  795.96  4973.6  794.97  4974.3  792.72  4980.4  792.72
  4981.6  789.72  5018.4  789.72  5019.6  792.72  5020.3  793.37  5021.7  796.44
  5050.1  795.19  5061.9  797.18  5083.5  804.12  5107.5  817.97  5120.2  822.52
  5138.2  826.37  5150.1  826.69  5164.2  828.77  5176.2  829.94  5193.6  830.45
#Mann= 5 ,-1 , 0
    4690      .1       0  4925.7     .13       0  4980.4    .045       0
  5019.6     .13       0  5138.2     .07       0
Bank Sta=4980.4,5019.6
Exp/Cntr=0.3,0.1

Type RM Length L Ch R = 1 ,29770   ,329,329,329
BEGIN DESCRIPTION:
North Deep Creek 81.0
END DESCRIPTION:
XS GIS Cut Line= 4
      1523695.63       869737.02      1523571.97       869737.02
      1523477.42       869693.38      1523350.19        869664.3
#Sta/Elev= 30
  4788.9  846.47  4798.2  845.08  4814.8  840.49  4847.1  830.56  4853.9  828.04
  4858.6  825.93  4878.8  818.56  4903.6  806.87  4912.6  803.74  4923.6   799.4
  4925.5  798.11  4929.9  796.84  4958.6  793.64  4969.7  792.63  4975.5  792.63
    4977  789.63    5023  789.63  5024.5  792.63  5025.5   799.6  5026.5   801.3
  5036.8   802.2  5062.8  805.42  5083.3  809.21  5088.6  810.78  5103.7  813.77
  5109.3   814.5  5125.1  817.35  5129.6  817.51  5145.1  820.18  5147.2  820.31
#Mann= 4 ,-1 , 0
  4788.9     .13       0  4975.5    .045       0  5024.5     .13       0
  5036.8     .07       0
Bank Sta=4975.5,5024.5
Exp/Cntr=0.3,0.1

Type RM Length L Ch R = 1 ,29441   ,417,417,417
BEGIN DESCRIPTION:
North Deep Creek 80.0
END DESCRIPTION:
XS GIS Cut Line= 3
      1523684.69       869391.56      1523582.88       869377.02
      1523299.22       869384.29
#Sta/Elev= 28
  4844.5   822.6  4862.3  820.18  4873.1  818.57    4892   815.1  4903.6  811.83
    4919  807.98  4927.5  805.57  4942.6  801.72    4962  792.46  4975.5  792.46
    4977  789.46    5023  789.46  5024.5  792.46  5025.6  794.76    5046  801.65
  5065.5  802.81  5076.4  803.73    5093     805  5119.8  807.52  5127.3  808.71
    5133  809.48  5145.7  811.42  5169.6  815.97  5183.7   818.3    5199  821.14
  5212.7  823.19  5223.3  824.12  5231.1  825.15
#Mann= 4 ,-1 , 0
  4844.5     .13       0  4975.5    .045       0  5024.5     .13       0
  5076.4     .07       0
Bank Sta=4975.5,5024.5
Exp/Cntr=0.3,0.1

Type RM Length L Ch R = 1 ,29024   ,374,374,374
BEGIN DESCRIPTION:
North Deep Creek 79.0
END DESCRIPTION:
XS GIS Cut Line= 3
      1523681.03       868966.11      1523430.15       868958.83
      1523215.57       869020.66
#Sta/Elev= 30
  4836.3  833.31  4851.1     831  4866.5  827.64  4897.8  819.61    4903   817.7
  4913.9  814.32  4939.8  807.18  4953.6  802.78  4955.3  801.88  4961.4  800.55
  4969.3  797.91  4972.9  795.45  4975.5   792.2    4977   789.2    5023   789.2
  5024.5   792.2  5032.6  798.99  5039.7  800.98  5044.9  800.94  5063.3  799.98
  5067.7  800.32  5102.5  802.75  5115.4  803.87  5127.4  806.13  5138.3  809.06
  5161.1  813.95  5173.8  816.27  5208.1  821.42  5218.6  822.59  5310.6  831.02
#Mann= 4 ,-1 , 0
  4836.3     .13       0  4975.5    .045       0  5024.5     .13       0
  5067.7     .07       0
Bank Sta=4975.5,5024.5
Exp/Cntr=0.3,0.1

Type RM Length L Ch R = 1 ,28650   ,341,341,341
BEGIN DESCRIPTION:
North Deep Creek 78.0
END DESCRIPTION:
XS GIS Cut Line= 4
      1523811.97       868587.92       1523575.6       868580.65
      1523390.15       868598.83      1522942.86       868806.11
#Sta/Elev= 30
    4671  839.29  4717.5  834.14  4751.8  829.11  4783.2  825.87  4799.3   822.9
  4826.4  816.83  4835.6  815.26  4863.9  809.14  4899.2  802.74  4936.1  798.68
  4957.4  799.26  4963.8  798.18  4970.2   793.8  4971.9  792.01  4975.5  791.99
    4977  788.99    5023  788.99  5024.5  791.99  5026.7  791.99  5028.1  797.08
  5028.7  797.43  5068.5  799.66  5072.9  799.96  5095.8  798.96  5150.1  802.26
  5339.8  818.47  5441.8  825.26  5471.3  827.89  5555.1  833.35  5586.8  835.88
#Mann= 4 ,-1 , 0
    4671     .11       0  4975.5    .045       0  5024.5     .11       0
  5068.5     .07       0
Bank Sta=4975.5,5024.5
Exp/Cntr=0.3,0.1

Type RM Length L Ch R = 1 ,28309   ,384,384,384
BEGIN DESCRIPTION:
North Deep Creek 77.5
END DESCRIPTION:
XS GIS Cut Line= 4
      1523778.75       868118.49      1523631.57       868142.45
      1523169.36        868409.5      1522874.92       868724.48
#Sta/Elev= 30
  4629.3  820.46  4662.4  816.62    4702  813.54  4762.4  804.99    4802  798.03
  4833.7   796.7  4870.3  799.89    4956  800.87  4968.5  799.79  4971.6  798.93
  4975.5   791.8    4977   788.8    5023   788.8  5024.5   791.8  5031.3  796.32
    5075  797.54  5111.2  797.35  5183.7  798.88  5198.7  798.49  5287.9  800.42
  5412.6  805.31  5463.9   808.6  5517.6   813.4  5547.1  816.72  5585.6  822.26
    5599  823.03  5611.6  825.43  5651.3   829.6  5702.4  834.07  5743.4  836.29
#Mann= 4 ,-1 , 0
  4629.3     .11       0  4975.5    .045       0  5024.5     .11       0
    5075     .07       0
#XS Ineff= 2 , 0
       0  4945.8  810.14  5081.1       0  810.14
Permanent Ineff=
       F       F
Bank Sta=4975.5,5024.5
Exp/Cntr=0.3,0.1

Type RM Length L Ch R = 1 ,27925   ,440,440,440
BEGIN DESCRIPTION:
North Deep Creek 77.0
END DESCRIPTION:
XS GIS Cut Line= 5
      1523797.47       868042.48      1523324.69        867926.1
      1523142.87       867940.65      1522801.05       868042.46
      1522502.89       868344.27
#Sta/Elev= 30
  4433.1   816.5  4531.5   803.9  4601.3  797.74  4652.3  795.98  4680.4  797.63
    4736  798.38  4820.6  797.48  4848.5  796.59  4905.6  797.67  4927.6  795.65
  4934.6  796.83  4944.2  797.03  4958.2  795.65  4975.5  789.05    4977  786.05
    5023  786.05  5024.5  789.05  5034.9  797.48  5056.1  797.56    5116  797.45
    5259  799.05  5346.7  797.79  5417.8  799.46  5477.6  802.01  5593.8  809.78
  5634.2  809.62  5660.3  811.94  5694.8  813.13  5710.5  814.69  5883.3  821.74
#Mann= 4 ,-1 , 0
  4433.1     .11       0  4975.5    .045       0  5024.5     .11       0
  5056.1     .07       0
#XS Ineff= 2 , 0
       0  4888.3  810.06  5111.7       0  810.06
Permanent Ineff=
       F       F
Bank Sta=4975.5,5024.5
Exp/Cntr=0.3,0.1

Type RM Length L Ch R = 1 ,27485   ,509,509,509
BEGIN DESCRIPTION:
North Deep Creek 76.0
END DESCRIPTION:
XS GIS Cut Line= 5
      1523924.68       867944.27      1523473.79       867620.64
      1523382.88       867493.37       1523295.6       867257.01
      1523310.15       867049.69
#Sta/Elev= 30
  4365.2  819.88    4441  812.73  4506.3   802.7  4544.9  800.24    4698  795.66
    4745   796.6  4753.9     797  4784.2  791.84  4824.2  793.17  4839.6  791.83
  4851.2  793.66  4865.6  791.54  4894.4  796.06    4933  797.42    4956  796.38
  4965.1  788.84  4969.2  788.82    4971  785.82    5029  785.82  5030.8  788.82
  5037.4     790    5051  794.53    5062  795.03  5242.8  795.34  5263.9  797.01
    5279  794.84  5338.7  800.52  5399.1  813.14  5475.4  824.06  5536.4  827.53
#Mann= 6 ,-1 , 0
  4365.2     .11       0    4745     .14       0  4969.2    .045       0
  5030.8     .14       0  5037.4     .07       0  5338.7     .09       0
#XS Ineff= 2 , 0
       0  4909.3  808.79               0
Permanent Ineff=
       F       F
Bank Sta=4969.2,5030.8
Exp/Cntr=0.3,0.1

Type RM Length L Ch R = 1 ,26976   ,272,272,272
BEGIN DESCRIPTION:
North Deep Creek 74.0
END DESCRIPTION:
XS GIS Cut Line= 5
      1523997.45       867482.49      1523877.42       867315.19
      1523677.42       867198.82      1523477.42       867093.37
      1523371.99       867038.83
#Sta/Elev= 30
  4627.7  815.21  4663.5   814.4  4700.2  811.03  4756.8  801.66  4788.2  797.42
  4848.9  792.58  4962.1  796.32  4967.8   793.8  4969.4  788.31  4976.9   788.3
  4978.2   785.3  5021.8   785.3  5023.1   788.3  5027.1   794.3  5035.6  794.37
  5073.3  794.96  5123.7  794.15  5138.2  795.02    5168  795.13  5184.2   794.2
    5190  795.16  5208.1  795.55  5262.7  795.02  5287.4  797.68  5303.8  801.49
  5311.6  803.67    5336  813.53  5361.8   820.5  5384.6   825.4  5409.8  828.29
#Mann= 5 ,-1 , 0
  4627.7     .07       0  4788.2     .14       0  4976.9    .045       0
  5023.1     .14       0  5035.6     .09       0
Bank Sta=4976.9,5023.1
Exp/Cntr=0.3,0.1

Type RM Length L Ch R = 1 ,26704   ,545,545,545
BEGIN DESCRIPTION:
North Deep Creek 73.0
END DESCRIPTION:
XS GIS Cut Line= 4
      1524015.62       867460.69       1523884.7         867097.
       1523884.7       866475.18       1523884.7       866322.44
#Sta/Elev= 30
  4535.2  815.23  4564.6  814.54  4588.2  812.46  4677.3  797.45  4704.1  795.02
  4733.8  793.88  4809.7  792.53  4870.2  794.57  4900.5  794.34  4921.7  792.82
  4950.6  793.35  4958.2  792.12  4960.9  787.79    4964  787.78  4966.1  784.78
  5033.9  784.78    5036  787.78  5044.4  787.78  5044.9  788.71  5062.5   794.3
  5075.8   795.4    5207  795.39  5240.6  793.77  5285.2  795.13  5492.2     797
  5540.6  799.01  5555.1  801.53  5604.3  817.91  5632.6  825.93  5696.3  840.07
#Mann= 4 ,-1 , 0
  4535.2     .07       0  4733.8     .14       0    4964    .045       0
    5036     .09       0
#XS Ineff= 2 , 0
       0                  5215.7       0  818.12
Permanent Ineff=
       F       F
Bank Sta=4964,5036
Exp/Cntr=0.3,0.1

Type RM Length L Ch R = 1 ,26159   ,675,675,675
BEGIN DESCRIPTION:
North Deep Creek 72.0
END DESCRIPTION:
XS GIS Cut Line= 4
      1524066.52       867515.19      1524281.06       867184.28
      1524397.43       866558.82      1524390.15       866340.61
#Sta/Elev= 30
  4669.4  815.11  4741.2  814.16  4821.6  810.19  4876.4  806.58    4932  800.15
  4946.1  799.62  4956.2  786.87  4958.9  786.87  4961.3  783.87  5038.7  783.87
  5041.1  786.87  5045.9  786.87  5056.4  792.81  5059.2  793.03  5092.4  788.83
  5102.2  791.01  5146.2  794.02  5260.2  793.65  5306.8  791.12  5334.3  792.78
  5554.8  793.34  5633.7  795.89  5683.6  794.77  5696.7  792.92    5740  794.31
  5763.7  796.25  5786.9  802.31  5804.4  808.95  5865.8  823.56  5918.3  832.71
#Mann= 5 ,-1 , 0
  4669.4     .07       0    4932     .14       0  4958.9    .045       0
  5041.1     .14       0  5865.8     .14       0
#XS Ineff= 2 , 0
       0                  5424.5       0  812.64
Permanent Ineff=
       F       F
Bank Sta=4958.9,5041.1
Exp/Cntr=0.3,0.1

Type RM Length L Ch R = 1 ,25484   ,526,526,526
BEGIN DESCRIPTION:
North Deep Creek 71.0
END DESCRIPTION:
XS GIS Cut Line= 4
      1524350.16       868013.37      1524582.88       867835.19
      1524808.34       867464.28      1525022.88       866987.92
#Sta/Elev= 30
  4229.5  819.68  4390.2  809.69  4447.4  807.98  4496.2  808.52  4576.7  801.32
  4592.1  795.96  4627.6  791.83  4761.4  790.78    4932  791.97  4969.9     792
  4971.6  791.63  4974.3  785.95  4975.8  782.95  5024.2  782.95  5025.7  785.95
  5026.7  789.55  5028.2  790.22  5039.2  791.84  5101.3  791.94  5116.2  788.96
  5123.8  791.44  5137.1  789.22  5150.7  791.57  5190.3  792.28  5201.3  791.43
  5367.3  791.86  5376.2  793.76    5402  802.88  5432.8  811.91  5479.1  822.62
#Mann= 4 ,-1 , 0
  4229.5     .07       0    4932     .14       0  4974.3    .045       0
  5025.7     .14       0
#XS Ineff= 2 , 0
       0                  5233.8       0  808.26
Permanent Ineff=
       F       F
Bank Sta=4974.3,5025.7
Exp/Cntr=0.3,0.1

Type RM Length L Ch R = 1 ,24958   ,692,692,692
BEGIN DESCRIPTION:
North Deep Creek 70.0
END DESCRIPTION:
XS GIS Cut Line= 4
      1524528.33       868344.29      1525095.61       867838.83
      1525161.07       867773.37      1525332.02       867689.71
#Sta/Elev= 30
  4210.7  822.66    4232  820.75  4255.6  816.23  4271.1  810.67  4331.9  796.57
  4360.1  793.88  4388.2  793.08  4403.5  791.52  4410.7  792.23    4426  791.33
  4443.4  792.81  4592.4  792.62  4923.5  789.73  4952.5  789.74  4958.8  790.63
  4967.8  787.88  4968.9  784.94  4974.3  784.94  4975.8  781.94  5024.2  781.94
  5025.7  784.94  5027.6  789.55    5033  792.01  5055.8  791.02    5077  792.02
  5095.9  800.46  5131.5  808.74  5180.1   812.3  5243.7  819.39  5253.4  819.62
#Mann= 4 ,-1 , 0
  4210.7     .07       0  4923.5     .14       0  4974.3    .045       0
  5025.7     .14       0
#XS Ineff= 2 , 0
       0  4706.2  805.64               0
Permanent Ineff=
       F       F
Bank Sta=4974.3,5025.7
Exp/Cntr=0.3,0.1

Type RM Length L Ch R = 1 ,24266   ,442,442,442
BEGIN DESCRIPTION:
North Deep Creek 69.0
END DESCRIPTION:
XS GIS Cut Line= 5
      1525233.82       868675.16      1525408.34       868464.29
      1525684.71       868242.47      1525862.89       868140.65
      1525975.63       868009.72
#Sta/Elev= 30
  4528.1  814.54  4553.2  812.13  4628.9  807.84  4674.5  803.93  4805.3  794.96
  4834.1  793.49  4930.2  791.04  4948.8  791.13  4974.3  784.86  4975.8  781.86
  5024.2  781.86  5025.7  784.86  5030.9  784.86  5034.8  786.01  5038.8  785.93
  5056.5  789.38  5060.5  789.36  5136.8  788.62  5256.2   788.9  5281.2  788.36
  5293.2  787.26    5349  789.49  5393.5  789.92  5410.5  791.97  5428.6  795.34
  5446.3  800.24  5481.9  811.43  5499.3  815.06  5516.6  817.53  5534.2  818.52
#Mann= 6 ,-1 , 0
  4528.1     .07       0  4930.2     .14       0  4974.3    .045       0
  5025.7     .14       0  5060.5     .07       0    5349     .14       0
#XS Ineff= 2 , 0
       0                    5150       0     807
Permanent Ineff=
       F       F
Bank Sta=4974.3,5025.7
Exp/Cntr=0.3,0.1

Type RM Length L Ch R = 1 ,23824   ,353,353,353
BEGIN DESCRIPTION:
North Deep Creek 68.0
END DESCRIPTION:
XS GIS Cut Line= 5
      1525633.79       869075.22      1525691.98       868922.47
      1525801.07       868726.11      1525859.25        868635.2
      1525950.17       868402.45
#Sta/Elev= 30
  4572.1  841.76  4584.4  840.69  4600.2  838.13  4622.7   832.9  4663.5  821.39
  4712.2   803.1    4728  796.88  4745.1  787.78  4760.4  785.73    4765  785.93
  4773.5  787.18    4787  788.15  4803.2  788.66  4840.3  788.98  4881.8  788.58
  4942.1  789.77  4968.8  786.24  4974.3  784.82  4975.8  781.82  5024.2  781.82
  5025.7  784.82  5031.6  784.83  5032.6  791.13    5037  791.54  5047.6  790.86
    5106  796.29    5196  804.01  5243.5  805.24  5299.2  808.12    5318  808.43
#Mann= 5 ,-1 , 0
  4572.1     .14       0  4712.2     .07       0  4942.1     .14       0
  4974.3    .045       0  5025.7     .14       0
#XS Ineff= 2 , 0
       0  4826.8  815.66               0
Permanent Ineff=
       F       F
Bank Sta=4974.3,5025.7
Exp/Cntr=0.3,0.1

Type RM Length L Ch R = 1 ,23471   ,284,284,284
BEGIN DESCRIPTION:
North Deep Creek 67.0
END DESCRIPTION:
XS GIS Cut Line= 4
       1526342.9       868769.75       1526193.8       868671.56
      1526048.35       868504.29      1525982.88       868409.73
#Sta/Elev= 30
  4748.3  808.41  4768.8  805.93  4802.9  799.92  4814.5  799.34  4828.5  797.54
  4855.8   795.8  4861.2  794.97    4881  793.76  4894.1  792.36    4916  791.39
  4938.1  789.54  4944.6   789.5  4972.8  784.14    4976  782.57  4976.9  782.57
  4978.2  779.57  5021.8  779.57  5023.1  782.57  5023.6   786.6  5031.6  789.11
  5052.7  787.63  5066.3  787.41  5095.5  788.77  5125.4  788.13  5156.6  788.36
  5173.9  790.19  5199.5  793.79  5213.4  797.68    5258  806.13  5263.5  806.55
#Mann= 4 ,-1 , 0
  4748.3     .14       0  4976.9    .045       0  5023.1     .14       0
  5125.4     .14       0
Bank Sta=4976.9,5023.1
Exp/Cntr=0.3,0.1

Type RM Length L Ch R = 1 ,23187   ,215,215,215
BEGIN DESCRIPTION:
North Deep Creek 66.0
END DESCRIPTION:
XS GIS Cut Line= 4
      1526397.44       868722.49      1526408.35       868500.65
      1526342.89       868398.83      1526171.96       868184.25
#Sta/Elev= 30
  4725.9  811.98  4790.9  805.33  4822.1  801.13  4882.9  795.65    4917  789.62
  4930.7  788.73    4939  790.02  4942.6   789.8  4948.9  788.27  4966.4   786.2
  4974.3  781.14  4975.8  778.14  5024.2  778.14  5025.7  781.14  5025.9  781.21
  5026.1  788.25    5028  788.54  5045.5  789.13  5055.4  788.37  5067.8  789.83
  5105.6  790.95  5158.6  788.72  5223.1   787.2  5235.2  785.89  5264.9  787.76
  5278.1  793.09  5299.9  811.49  5309.9  816.54  5322.1   820.7  5343.4   824.7
#Mann= 4 ,-1 , 0
  4725.9     .14       0  4974.3    .045       0  5025.7     .14       0
  5158.6     .14       0
Bank Sta=4974.3,5025.7
Exp/Cntr=0.3,0.1

Type RM Length L Ch R = 1 ,22972   ,402,402,402
BEGIN DESCRIPTION:
North Deep Creek 65.0
END DESCRIPTION:
XS GIS Cut Line= 6
       1526422.9       868726.08      1526455.62       868562.47
      1526550.17        868486.1      1526619.26       868442.47
       1526753.8       868442.47      1526913.79       868449.74
#Sta/Elev= 30
  4682.6   813.4  4743.9  804.18  4779.3   800.7  4802.8  799.11  4818.2  798.87
  4843.1  796.84  4878.6  795.35  4936.9  790.92  4952.1  790.41  4967.2  788.69
    4976     781  4976.9     781  4978.2     778  5021.8     778  5023.1     781
  5026.6  782.12  5065.1  787.07  5115.9  785.65  5148.6  786.08    5175  784.91
  5186.7  785.77  5189.3  785.45  5193.3  786.75  5206.8  789.16  5225.8  788.14
  5230.5  790.06  5252.4  796.05  5296.9  804.55  5311.9   806.9  5347.4  810.44
#Mann= 3 ,-1 , 0
  4682.6     .14       0  4976.9    .045       0  5023.1     .14       0
Bank Sta=4976.9,5023.1
Exp/Cntr=0.3,0.1

Type RM Length L Ch R = 1 ,22570   ,171,171,171
BEGIN DESCRIPTION:
North Deep Creek 64.0
END DESCRIPTION:
XS GIS Cut Line= 4
      1526576.01       868887.12      1526653.05       868760.44
      1526781.44       868614.93      1526855.04       868488.28
#Sta/Elev= 30
  4891.8  824.58  4906.8  822.27  4922.3  818.78  4937.3  813.11  4952.9  806.52
  4962.1  800.58    4969  794.13  4980.6  787.22  4980.9  780.73    4982  780.72
  4983.1  777.72  5016.9  777.72    5018  780.72  5024.1  780.72  5027.5  781.83
  5050.1  786.98    5067  787.46  5073.4   788.1  5100.5  788.25    5134  786.23
  5158.8  788.22  5186.4  789.49  5212.2  791.54  5238.1  795.57  5251.3  796.78
  5283.1  797.58  5304.7  799.79  5337.3  801.84  5357.5  804.54  5380.6   805.6
#Mann= 3 ,-1 , 0
  4891.8     .14       0    4982    .045       0    5018     .14       0
Bank Sta=4982,5018
Exp/Cntr=0.3,0.1

Type RM Length L Ch R = 1 ,22399   ,381,381,381
BEGIN DESCRIPTION:
North Deep Creek 63.0
END DESCRIPTION:
XS GIS Cut Line= 5
      1526855.63       868915.21      1526797.44       868824.29
      1526797.44       868671.56      1526844.71       868558.83
       1526862.9       868500.62
#Sta/Elev= 30
  4889.3  808.54  4905.9   806.6  4915.4   804.3  4941.2  794.96  4954.6  788.87
  4973.9  787.03  4976.4  780.34  4977.8  777.34  5022.2  777.34  5023.6  780.34
  5029.3  783.92    5033  785.66  5053.7  787.41  5063.4  786.11  5066.9  786.19
  5085.7   787.7  5109.2  788.33  5120.9  789.41  5137.1  789.54  5146.7  791.25
  5162.3  791.07  5188.8  793.62  5199.1  793.98    5218  796.25  5259.5  798.43
  5286.6  800.74  5298.7  802.53  5310.3  803.35  5321.1  804.94  5333.2  806.05
#Mann= 3 ,-1 , 0
  4889.3     .14       0  4976.4    .045       0  5023.6     .14       0
Bank Sta=4976.4,5023.6
Exp/Cntr=0.3,0.1

Type RM Length L Ch R = 1 ,22018   ,355,355,355
BEGIN DESCRIPTION:
North Deep Creek 61.0
END DESCRIPTION:
XS GIS Cut Line= 4
      1527140.92       868715.89       1527106.7       868633.76
       1527048.5       868541.32      1527026.22       868493.35
#Sta/Elev= 30
    4819  808.82  4833.7  805.91  4836.8  805.33  4841.7  804.58  4848.6  803.21
  4853.9   802.1    4864  799.61  4882.6  795.91  4887.8  795.07  4911.4  792.04
    4917  790.99  4936.3  788.24    4949   787.1  4955.8  786.19  4960.2  786.73
  4966.2  786.55  4968.1  785.27  4973.4  779.37  4984.3  779.41  4985.2  776.41
  5014.8  776.41  5015.7  779.41  5016.9  779.37  5017.2  781.39  5017.8  784.88
  5022.5  796.55  5031.6  797.09  5044.2  800.61  5055.3  804.56  5070.1  808.62
#Mann= 3 ,-1 , 0
    4819     .14       0  4984.3    .045       0  5015.7     .14       0
Bank Sta=4984.3,5015.7
Exp/Cntr=0.3,0.1

Type RM Length L Ch R = 1 ,21663   ,395,395,395
BEGIN DESCRIPTION:
North Deep Creek 60.0
END DESCRIPTION:
XS GIS Cut Line= 3
        1527292.       868755.19      1527375.63        868646.1
      1527437.46       868467.88
#Sta/Elev= 30
  4817.4  813.63  4821.7  812.74  4836.1  805.64  4854.5  801.74  4883.4  795.21
  4891.2  793.89  4911.3  791.58  4936.7  788.01  4947.9  785.44  4954.9  780.16
  4955.8  779.93  4956.1  779.14  4971.2  779.14  4972.8  776.14  5027.2  776.14
  5028.8  779.14  5031.2  779.15  5032.4     782  5033.5   789.8    5039  790.18
  5042.6  790.76  5046.5  792.84  5053.4  795.96    5060  799.82    5080  803.71
  5090.7  806.54  5095.7  807.56  5112.3  809.97  5134.8  813.78  5143.5  815.44
#Mann= 3 ,-1 , 0
  4817.4     .14       0  4971.2    .045       0  5028.8     .14       0
Bank Sta=4971.2,5028.8
Exp/Cntr=0.3,0.1

Type RM Length L Ch R = 1 ,21268   ,302,302,302
BEGIN DESCRIPTION:
North Deep Creek 59.0
END DESCRIPTION:
XS GIS Cut Line= 5
      1527822.89         869017.      1527768.36       868882.47
      1527768.36       868751.56      1527771.99       868682.47
      1527735.62       868471.54
#Sta/Elev= 30
  4678.4  818.46  4703.7  812.15  4714.6  810.27  4723.5  807.93  4777.8  797.39
  4810.3  793.04  4832.2  791.04  4882.6  787.55  4895.1  787.35    4929  785.28
  4936.6  785.75  4966.1  785.79  4967.6  781.51    4970  778.88  4973.8  778.88
  4975.3  775.88  5024.7  775.88  5026.2  778.88  5028.9   778.9  5032.6  788.64
  5033.7  789.82  5076.4  790.05  5092.1  791.06  5114.5  793.49  5127.4  796.41
  5152.3  801.04  5169.2  805.87  5190.5  810.58    5225  815.73  5237.7  817.08
#Mann= 3 ,-1 , 0
  4678.4     .14       0  4973.8    .045       0  5026.2     .14       0
Bank Sta=4973.8,5026.2
Exp/Cntr=0.3,0.1

Type RM Length L Ch R = 1 ,20966   ,302,302,302
BEGIN DESCRIPTION:
North Deep Creek 58.0
END DESCRIPTION:
XS GIS Cut Line= 4
      1528142.91       869006.13      1528070.18       868773.38
      1528073.81       868591.56      1528081.08       868257.05
#Sta/Elev= 30
  4722.2  820.59  4758.7  816.83    4779  814.05  4796.7  810.96  4848.2   799.1
  4879.2  794.08    4901   791.9  4941.3   786.1  4965.6  785.88  4976.4  778.73
  4977.8  775.73  5022.2  775.73  5023.6  778.73  5026.1  778.74  5026.5  781.13
  5043.1  787.51  5054.6  789.41  5119.7  790.21    5140  792.65  5155.3  796.57
  5177.8  797.01  5195.3  800.02  5303.5  804.73  5353.4  809.32  5363.6  809.33
  5394.1  811.52  5426.8  815.21  5450.7  819.23    5464  820.04  5482.5  823.21
#Mann= 3 ,-1 , 0
  4722.2     .14       0  4976.4    .045       0  5023.6     .14       0
Bank Sta=4976.4,5023.6
Exp/Cntr=0.3,0.1

Type RM Length L Ch R = 1 ,20664   ,395,395,395
BEGIN DESCRIPTION:
North Deep Creek 57.0
END DESCRIPTION:
XS GIS Cut Line= 4
      1528353.82        868987.9      1528375.63       868769.74
      1528364.72       868667.92      1528393.81       868533.38
#Sta/Elev= 30
  4704.4  816.58  4724.9  813.64  4747.5  811.48  4764.8   808.6  4785.7  804.47
    4802  799.52  4823.7  794.39  4827.2  793.67  4844.6  791.79  4853.4  790.08
  4880.3  788.01  4904.1  785.52  4916.2  785.01  4933.3  787.65  4957.7  787.04
    4971  784.12  4974.9  780.58  4976.4  778.55  4977.8  775.55  5022.2  775.55
  5023.6  778.55  5026.2   780.8  5039.2  785.16  5041.1   786.2  5076.1  786.82
  5078.8  787.56  5094.1  794.01  5125.7   810.6  5137.2  814.75  5163.7  822.41
#Mann= 3 ,-1 , 0
  4704.4     .14       0  4976.4    .045       0  5023.6     .14       0
Bank Sta=4976.4,5023.6
Exp/Cntr=0.3,0.1

Type RM Length L Ch R = 1 ,20269   ,474,474,474
BEGIN DESCRIPTION:
North Deep Creek 56.0
END DESCRIPTION:
XS GIS Cut Line= 4
      1528717.45       869053.39      1528761.09       868813.38
      1528761.09       868657.01      1528717.47       868562.51
#Sta/Elev= 30
  4595.4  803.06  4612.7  802.32  4639.3  799.87  4674.6  797.74    4738  793.53
  4746.7  792.83  4757.6  791.54  4778.4  790.56  4796.6  789.23  4814.5  788.72
  4833.3  787.54  4841.1  786.79  4852.2  786.22  4892.3  784.81  4911.3  784.41
  4925.4  783.37  4944.1  784.83  4954.1  785.31  4963.2  785.38  4970.7  780.92
  4970.9  778.36  4973.8  778.36  4975.3  775.36  5024.7  775.36  5026.2  778.36
  5028.8  778.37  5053.3  794.76  5078.2  808.16  5086.4  812.11  5099.8  816.61
#Mann= 3 ,-1 , 0
  4595.4     .14       0  4973.8    .045       0  5026.2     .14       0
Bank Sta=4973.8,5026.2
Exp/Cntr=0.3,0.1

Type RM Length L Ch R = 1 ,19795   ,161,161,161
BEGIN DESCRIPTION:
North Deep Creek 55.0
END DESCRIPTION:
XS GIS Cut Line= 4
      1529331.98       868529.74      1529193.82       868555.19
      1529008.36       868533.38      1528848.39       868500.66
#Sta/Elev= 30
  4844.8  808.22  4873.5   802.6  4907.1  795.27  4933.9  784.45  4963.1   781.2
  4966.7   779.1  4966.9  778.03  4979.8  775.03  5020.2  775.03  5021.4  778.03
  5031.3  783.43  5056.5  785.28  5069.2  784.89  5077.3  783.78  5105.9  784.78
  5127.6  782.97  5143.8  783.05    5172  781.53  5175.4  781.28  5185.6  779.16
  5196.4  779.63  5201.1  780.07    5206   782.1  5212.8  787.17  5224.8  788.05
  5236.4  790.74  5272.4  795.49  5288.2  796.45  5319.5  802.02  5335.3  806.02
#Mann= 3 ,-1 , 0
  4844.8     .14       0  4966.9    .045       0  5021.4     .14       0
Bank Sta=4966.9,5021.4
Exp/Cntr=0.3,0.1

Type RM Length L Ch R = 1 ,19634   ,197,197,197
BEGIN DESCRIPTION:
North Deep Creek 54.0
END DESCRIPTION:
XS GIS Cut Line= 4
      1529277.42       868340.67      1529099.27       868453.38
      1528997.45        868486.1      1528862.95        868475.2
#Sta/Elev= 30
  4889.8  828.86  4906.4   823.9  4911.7  821.83  4939.6  804.24  4946.2  801.59
  4954.3  797.31  4974.9  779.32  4977.4  777.95  4978.6  777.94  4979.8  774.94
  5020.2  774.94    5031  777.95  5033.5  784.47  5033.8  784.74  5047.1  783.89
  5061.7  783.61  5091.1  783.52  5122.3  784.11  5143.2   782.9  5160.7  783.42
  5167.4  782.59  5185.2   778.6  5203.8  780.49  5218.8  783.57  5231.6   786.8
    5243  788.29  5274.6   789.7  5295.7  792.05  5333.1  798.31  5342.5  800.61
#Mann= 3 ,-1 , 0
  4889.8     .14       0  4978.6    .045       0    5031     .14       0
Bank Sta=4978.6,5031
Exp/Cntr=0.3,0.1

Type RM Length L Ch R = 1 ,19437   ,192,192,192
BEGIN DESCRIPTION:
North Deep Creek 53.0
END DESCRIPTION:
XS GIS Cut Line= 3
      1529062.92       868235.17      1528961.09       868424.29
      1528870.16       868446.11
#Sta/Elev= 26
  4857.4  825.61  4885.4  822.01  4889.1  820.85  4964.2  784.47  4968.7  782.44
  4976.5  779.64  4980.5  777.79  4987.4  774.78  5012.7  774.78  5013.4  777.78
  5013.8  777.78  5014.4  778.93  5017.6  779.66  5022.9   779.5  5031.6  778.98
    5045  779.17    5047  779.43  5072.2  784.25  5083.7  784.74  5097.6  786.46
  5102.9  786.54  5111.1  786.39  5121.9  788.78  5152.3   794.1  5163.3  796.17
  5165.7  796.77
#Mann= 3 ,-1 , 0
  4857.4     .14       0  4980.5    .045       0  5013.4     .14       0
Bank Sta=4980.5,5013.4
Exp/Cntr=0.3,0.1

Type RM Length L Ch R = 1 ,19245   ,218,218,218
BEGIN DESCRIPTION:
North Deep Creek 52.0
END DESCRIPTION:
XS GIS Cut Line= 3
      1529015.68       868191.55      1528913.82       868202.47
      1528691.96       868315.21
#Sta/Elev= 26
  4855.4  814.49  4877.9  808.37  4882.1  807.29  4905.2  800.02  4915.6  797.86
  4927.2   793.2  4954.5  781.32  4961.7  779.04    4973  777.61  4975.9  777.61
  4977.2  774.61  5022.8  774.61  5024.1  777.61  5042.9  782.41  5047.4  783.15
  5058.7  783.68  5072.7  784.08  5100.5  791.43  5120.1  799.23  5138.8  806.06
  5151.4  810.54  5166.8     818  5187.5  821.16  5199.4  822.07  5204.7  823.04
  5206.7  823.28
#Mann= 3 ,-1 , 0
  4855.4     .14       0  4975.9    .045       0  5024.1     .14       0
Bank Sta=4975.9,5024.1
Exp/Cntr=0.3,0.1

Type RM Length L Ch R = 1 ,19027   ,308,308,308
BEGIN DESCRIPTION:
North Deep Creek 51.0
END DESCRIPTION:
XS GIS Cut Line= 3
      1529001.07       868031.55        1528892.        868006.1
      1528688.33       868013.37
#Sta/Elev= 30
  4846.9   807.7  4866.6  799.44  4875.8  796.37  4877.6  795.87  4898.2  793.13
  4903.8  791.83  4915.4  788.92  4924.7  786.76  4972.8  775.92  4978.6  775.91
  4979.8  772.91  5020.2  772.91  5021.4  775.91    5024     778  5030.8  779.58
  5034.8  779.79  5042.8  781.45  5049.4     783    5055  784.84  5059.9   786.6
  5069.6   791.8  5078.8   795.8  5099.1  804.97  5115.4  811.31  5118.7  812.72
  5135.8   817.9  5141.1  820.08  5148.2  823.34  5158.2  824.39  5162.7  825.18
#Mann= 3 ,-1 , 0
  4846.9     .14       0  4978.6    .045       0  5021.4     .14       0
Bank Sta=4978.6,5021.4
Exp/Cntr=0.3,0.1

Type RM Length L Ch R = 1 ,18719   ,313,313,313
BEGIN DESCRIPTION:
North Deep Creek 50.0
END DESCRIPTION:
XS GIS Cut Line= 2
      1529099.32       867766.11      1528852.04       867686.11
#Sta/Elev= 30
  4835.8  808.22  4844.5  807.04  4848.7  806.33  4855.4  805.55    4860  804.83
  4865.2  803.87  4868.8  802.96  4874.6  802.21    4885   800.3  4888.6  799.25
  4916.3  787.42  4925.7  784.05  4929.1  783.01  4939.2  780.71  4942.7  779.99
    4947  779.35  4959.7  776.62  4973.1  772.46  4975.9  772.46  4977.2  769.46
  5022.8  769.46  5024.1  772.46  5024.9  774.53  5031.7  779.91  5034.1   780.7
  5050.9  789.73  5053.8  791.94  5061.5   797.6  5091.3  820.46  5095.7  822.71
#Mann= 3 ,-1 , 0
  4835.8     .14       0  4975.9    .045       0  5024.1     .14       0
Bank Sta=4975.9,5024.1
Exp/Cntr=0.3,0.1

Type RM Length L Ch R = 1 ,18406   ,400,400,400
BEGIN DESCRIPTION:
North Deep Creek 49.0
END DESCRIPTION:
XS GIS Cut Line= 4
      1529168.37       867722.49      1529153.82       867580.64
      1529153.82       867493.37      1529193.82       867431.55
#Sta/Elev= 30
  4786.1  808.72    4803  806.19  4810.4   805.2  4826.2  802.67  4836.7  801.37
    4846  799.66  4855.2  798.29  4866.1  796.11    4870  795.15  4872.8  794.26
  4890.3  790.58  4901.8  787.29  4905.5  786.46  4914.8  784.72  4923.2  782.99
  4936.5  779.66  4960.8  774.89  4961.6  774.43  4963.9  771.68    4968  771.67
  4973.2  771.48  4974.7  768.48  5025.3  768.48  5026.8  771.48  5046.8  771.48
  5051.8  775.26  5062.1  782.16  5071.8   789.7    5077  793.33  5089.6  798.94
#Mann= 3 ,-1 , 0
  4786.1     .14       0  4973.2    .045       0  5026.8     .14       0
Bank Sta=4973.2,5026.8
Exp/Cntr=0.3,0.1

Type RM Length L Ch R = 1 ,18006   ,87,87,87
BEGIN DESCRIPTION:
North Deep Creek 48.0
END DESCRIPTION:
XS GIS Cut Line= 4
      1529284.71       867809.75      1529393.82       867749.74
      1529473.82       867738.83      1529577.42       867689.75
#Sta/Elev= 30
  4835.2  812.47  4843.5  810.68  4872.9  803.12  4903.3  794.62  4917.9  790.16
  4932.7  784.36    4947  780.45  4966.5  777.53  4977.2  770.68  4977.4  770.06
  4978.1  770.05  4978.6   768.7  4979.8   765.7  5020.2   765.7  5021.4   768.7
  5024.1   768.7  5027.3  769.77  5035.5  770.23  5051.9  770.36  5056.8  771.81
  5065.3   776.1  5074.2  779.74  5080.5  783.15  5085.2  785.95  5094.4  790.57
  5105.6   795.6    5118  801.97  5133.5  809.05  5149.6  810.37  5155.1  810.55
#Mann= 3 ,-1 , 0
  4835.2     .14       0  4978.6    .045       0  5021.4     .14       0
Bank Sta=4978.6,5021.4
Exp/Cntr=0.3,0.1

Type RM Length L Ch R = 1 ,17919   ,61,61,61
BEGIN DESCRIPTION:
North Deep Creek 47.5
END DESCRIPTION:
XS GIS Cut Line= 4
      1529333.48       867868.11        1529403.       867838.62
      1529491.47       867819.66      1529600.98       867769.12
#Sta/Elev= 30
  4888.1  798.18  4915.7   790.9    4942  783.13  4955.3  778.67    4962  772.72
    4972  768.05  4974.5  766.31  4975.9  766.01  4977.2  763.01  5022.8  763.01
  5028.3  766.13  5029.4  768.19  5037.6  769.35  5049.9  768.86  5067.9  769.51
  5074.4  769.47  5077.4  769.89    5080   769.9  5086.8  771.11  5099.1  776.83
  5111.5  779.25  5114.4  781.91  5117.7  785.68  5126.1  794.54  5133.3  794.62
  5140.8  795.45  5147.9  799.61  5161.9  802.17  5170.4  805.11  5174.7  805.25
#Mann= 3 ,-1 , 0
  4888.1     .14       0  4975.9    .045       0  5028.3     .14       0
#XS Ineff= 2 , 0
       0                    5050       0     780
Permanent Ineff=
       F       F
Bank Sta=4975.9,5028.3
Exp/Cntr=0.3,0.1

Type RM Length L Ch R = 1 ,17858   ,333,333,333
BEGIN DESCRIPTION:
North Deep Creek 47.0
END DESCRIPTION:
XS GIS Cut Line= 5
        1529327.        867924.9      1529408.65       867905.91
      1529490.89       867876.18      1529531.38       867842.02
      1529599.03        867814.2
#Sta/Elev= 30
  4871.4  808.25  4888.6  802.56  4908.7  792.18    4918  787.95    4924  785.57
    4937  779.83    4941  778.32  4955.3  769.13  4969.2  761.95  4971.8  757.97
  4973.2  754.44  4974.7  751.44  5025.3  751.44  5026.8  754.44  5031.1  757.13
  5031.2  758.24  5040.8  763.41  5043.3  764.57  5049.5     766  5065.4   766.7
  5090.8  768.13  5096.3  768.89  5107.5  770.97    5124  780.56    5145  785.85
  5146.3  785.94    5148  786.39  5157.9  788.18  5164.7  791.27  5168.8  794.01
#Mann= 3 ,-1 , 0
  4871.4     .14       0  4973.2    .045       0  5026.8     .14       0
Bank Sta=4973.2,5026.8
Exp/Cntr=0.3,0.1

Type RM Length L Ch R = 1 ,17525   ,317,317,317
BEGIN DESCRIPTION:
North Deep Creek 46.0
END DESCRIPTION:
XS GIS Cut Line= 4
      1529448.35       868289.75      1529528.36       868220.65
      1529642.91       868162.47      1529753.82       868084.28
#Sta/Elev= 30
  4853.7  817.01  4854.8   816.7  4878.8   808.2  4895.8  801.68  4914.9  791.52
  4933.3  783.51  4959.2  771.74  4972.2  762.06  4975.9  751.94  4977.2  748.94
  5022.8  748.94  5024.1  751.94  5033.6  751.94  5035.7  752.59  5047.6  754.35
  5068.6  754.78    5080   755.8  5087.9   756.9  5104.3   759.8  5122.9  762.54
  5129.4  763.85    5142  766.06  5148.7  766.78  5156.7  767.96  5159.9  769.89
  5173.2  777.46  5183.9  778.13  5190.4  779.08  5207.4  780.57  5223.6  783.34
#Mann= 3 ,-1 , 0
  4853.7     .14       0  4975.9    .045       0  5024.1     .14       0
Bank Sta=4975.9,5024.1
Exp/Cntr=0.3,0.1

Type RM Length L Ch R = 1 ,17208   ,135,135,135
BEGIN DESCRIPTION:
North Deep Creek 45.0
END DESCRIPTION:
XS GIS Cut Line= 4
      1529699.26       868560.69      1529744.73       868469.74
      1529879.28       868309.74      1529970.22       868249.72
#Sta/Elev= 30
  4857.4  803.86  4879.3  795.32  4893.9  788.81  4904.1  785.31  4921.2  775.55
  4928.3  770.79  4933.5  769.38  4948.6   766.3  4959.1  760.37    4965  756.65
  4973.2  750.28  4974.7  747.28  5025.3  747.28  5026.8  750.28  5034.1  752.82
  5051.2  755.08  5067.5   755.4  5088.2  758.43  5100.2  762.47    5124  771.44
  5132.3  772.52  5160.6  773.94  5176.7   772.4  5186.1   776.5  5190.6  778.91
  5205.8  785.81  5223.7   787.3  5241.7  791.97  5268.5  790.95  5277.1  791.92
#Mann= 3 ,-1 , 0
  4857.4     .14       0  4973.2    .045       0  5026.8     .14       0
Bank Sta=4973.2,5026.8
Exp/Cntr=0.5,0.3

Type RM Length L Ch R = 1 ,17073   ,127,127,127
BEGIN DESCRIPTION:
Styers Mill Rd (NDC) us
END DESCRIPTION:
XS GIS Cut Line= 5
      1529907.63       868763.73      1529966.77       868721.49
      1529840.05       868416.31      1529878.06       868340.28
      1529924.73       868299.04
#Sta/Elev= 30
  4703.8   811.7  4713.9   808.4  4719.6  805.73  4734.9  801.56  4770.2  784.06
  4790.5  779.77    4814   778.3  4841.8  777.46  4860.7  775.45  4887.8  773.61
  4893.7  771.96  4901.3  770.66  4902.9  770.88  4916.6  767.44  4949.3  757.48
  4962.5   751.7    4975     745    5025     745  5037.5   751.7  5072.4   752.8
  5093.8  755.82  5098.5  755.65  5106.9  756.83  5116.5  758.71  5139.7  766.53
  5163.4  772.79  5209.6  773.93  5218.7  773.42  5234.9  783.35  5254.2  787.23
#Mann= 3 ,-1 , 0
  4703.8     .14       0  4962.5    .045       0  5037.5     .14       0
#XS Ineff= 2 , 0
       0  4836.5  783.06  5163.5       0  772.99
Permanent Ineff=
       F       F
Bank Sta=4962.5,5037.5
Exp/Cntr=0.5,0.3

Type RM Length L Ch R = 3 ,16997   ,,,
BEGIN DESCRIPTION:
Styers Mill Rd (NDC) tor
Structure ID: LDS_NDC_04
Approximate Survey Structure
END DESCRIPTION:
Bridge Culvert--1,0,-1,-1, 0
Deck Dist Width WeirC Skew NumUp NumDn MinLoCord MaxHiCord MaxSubmerge Is_Ogee
54.5,43,3,0, 12, 12, , , 0.95, 0, 1,1,,
    4754  4780.2  4884.5    4891    4891    5109    5109  5115.6  5174.1  5193.1
  5227.7  5273.3
  788.06   786.7  780.82   780.6   780.6  773.33  773.33  773.11  772.64   773.4
  775.96  787.32
     725     725     725     725   775.2   767.9     725     725     725     725
     725     725
    4754  4780.2  4884.5    4891    4891    5109    5109  5115.6  5174.1  5193.1
  5227.7  5273.3
  788.06   786.7  780.82   780.6   780.6  773.33  773.33  773.11  772.64   773.4
  775.96  787.32
     725     725     725     725   775.2   767.9     725     725     725     725
     725     725
Pier Skew, UpSta & Num, DnSta & Num=  ,4945.5, 2 ,4945.5, 2 , 0 , 0 , 0 ,0,0
       4       4
   758.3     775
       4       4
  759.29     775
Pier Skew, UpSta & Num, DnSta & Num=  ,5054.5, 2 ,5054.5, 2 , 0 , 0 , 0 ,0,0
       4       4
  750.75     772
       4       4
  753.45     772
Abutment Skew #Up #Dn= , 2 , 2
    4891    4923
   775.2   765.4
    4891    4923
   775.2  768.66
Abutment Skew #Up #Dn= , 2 , 2
    5077    5109
  753.69   767.9
    5077    5109
  752.84  767.89
BR Coef= 1 , 1 , 0 ,1.25, 0 ,,,0.8,0,2,0,
WSPro=,,,, 1 ,,,, 0 ,,,, 0 ,,,,-1 ,-1 ,-1 , 0 , 0 , 0 , 0 , 0
BC Design=,, 0 ,, 0 ,,,,,,
BC HTab HWMax=811.7
